HEC-RAS study dtl_little_ivy_crk.prj: dtl_Little_Ivy_Crk

--- dtl_little_ivy_crk.g01 (geometry) --- (continued)

Type RM Length L Ch R = 1 ,11892   ,427.63,438.16,448.17
XS GIS Cut Line= 3
  955074.0739713   766552.120733  954601.4191227  766832.0004134
  954372.9452664   767266.100638
#Sta/Elev= 30
       0 2067.19   15.94 2061.56    52.9 2051.16   77.02 2046.77   88.81 2043.37
  114.59 2040.12  224.16 2034.65  428.89 2036.25  522.36 2035.37  551.32 2035.89
  578.13 2033.44  599.06 2030.55  620.85 2028.73  624.33 2030.84  631.04 2035.04
   634.3 2036.26  651.38 2035.59  715.32  2036.6   809.8 2036.43  887.57 2039.31
  913.01 2041.76  919.19 2043.01  934.64 2048.24  942.37 2051.81  962.41 2053.35
  974.83 2055.68  984.67 2065.26  996.76 2073.87 1020.65 2087.24 1039.86 2099.04
#Mann= 5 ,-1 , 0
       0     .09       0  114.59     .05       0  551.32     .07       0
  599.06    .055       0  624.33     .05       0
Bank Sta=599.06,624.33
Exp/Cntr=0.3,0.1

Type RM Length L Ch R = 1 ,11454   ,478.71,506.89,537.63
XS GIS Cut Line= 3
  954964.1209472  766497.8589729  954420.0687224   766516.422045
   954087.353714  766676.3534372
#Sta/Elev= 30
       0 2057.26   63.27 2046.37   83.85 2039.19   89.88 2036.23   98.96 2033.91
  168.52 2032.85  221.38 2034.02  300.95 2033.09  372.24 2033.97  571.87 2032.34
  633.99 2033.74  649.33 2035.56  654.59 2036.34  661.88 2034.23  691.82 2028.38
  702.35 2027.67  712.06 2028.72   725.5 2034.27  737.42 2041.54  740.01 2042.44
  756.85 2044.73     766 2044.62  773.78 2046.52  776.21 2048.68   809.6 2067.92
  827.41 2078.84   837.2 2082.39  847.93 2088.37  894.77 2107.18  913.53 2113.03
#Mann= 6 ,-1 , 0
       0     .07       0  168.52     .05       0  649.33     .07       0
  691.82    .055       0  712.06     .05       0   809.6     .08       0
#XS Ineff= 2 , 0
       0     222  2038.6               0
Permanent Ineff=
       F       F
Bank Sta=691.82,712.06
Exp/Cntr=0.3,0.1

Type RM Length L Ch R = 1 ,10947   ,619.9,613.88,609.02
XS GIS Cut Line= 5
  954937.5983231  766459.0043169  954439.0393465  766396.6847008
  954298.4892023  766307.8455327  954234.8435062  766274.6966046
   954127.441266  765990.9431322
#Sta/Elev= 30
       0 2061.12   16.69 2058.33   41.07 2052.43   56.95 2046.64   70.37 2040.75
   91.47 2033.63  106.74 2032.26  121.31  2032.1  159.11 2033.19  263.34 2032.36
  355.76 2033.15  413.44 2032.19  482.28 2032.04  586.13  2033.6  795.45 2033.26
  828.75 2033.81  848.37 2032.41  861.55 2032.79  881.57  2029.2  887.73 2027.84
  903.59 2027.51  917.27  2028.4  918.51 2029.47  928.83 2036.37  952.91 2042.59
  970.68 2042.35  982.44 2047.81  995.07 2052.56 1008.02 2060.61 1043.88 2080.75
#Mann= 5 ,-1 , 0
       0     .07       0  121.31     .05       0  795.45     .07       0
  881.57    .055       0  918.51     .09       0
#XS Ineff= 2 , 0
       0     334  2037.5               0
Permanent Ineff=
       F       F
Bank Sta=881.57,918.51
Exp/Cntr=0.3,0.1

Type RM Length L Ch R = 1 ,10333   ,60.44,51.92,28.22
XS GIS Cut Line= 6
  954974.9057152  766359.0701087   954808.499571  766164.9995805
  954794.7001469  766099.2997404  954772.1997949  766074.5005083
  954747.3002109  766031.7003803  954708.2940028  765992.3286042
#Sta/Elev= 30
       0 2061.56   17.22 2051.79   23.94 2048.83   35.96 2044.56   47.77 2039.68
   50.71 2038.09   58.84 2036.87   66.48 2036.18   78.48 2033.65   85.55  2032.8
  116.15 2031.67  172.64 2030.31  202.09 2030.27  249.21 2029.78  255.63  2029.3
  307.71  2027.4  317.96  2023.2  320.54  2022.8  322.99  2022.3  339.24    2022
  356.51    2021   360.2  2023.6  373.22  2025.7  394.92    2037  406.14  2037.9
  426.17  2035.8  433.91 2041.26  439.33 2044.84  454.81 2056.38  461.67  2061.2
#Mann= 5 ,-1 , 0
       0     .07       0   85.55     .05       0  307.71     .07       0
  320.54     .05       0   360.2     .07       0
Bank Sta=320.54,360.2
Exp/Cntr=0.5,0.3

Type RM Length L Ch R = 1 ,10281   ,33.4,36.74,50.66
XS GIS Cut Line= 6
  955009.7442432  766120.5323804  954942.6886272  766146.3228444
  954918.3000191  766142.2002204  954873.9997311  766102.7997724
   954800.800115  766058.7001883  954715.0247548  765985.6869402
#Sta/Elev= 29
       0 2039.23   5.709 2039.17  25.819 2036.53  30.765 2036.84  40.183 2036.58
  45.688 2036.13  47.649 2036.28  65.094 2035.95  67.383 2035.46  69.392 2035.19
  73.642 2034.28  91.454  2031.3  93.299  2030.8 143.836    2029 163.068  2027.2
 167.675  2025.4  178.03    2023 179.894  2021.8 182.434  2021.1 194.441  2020.7
 235.039  2022.7 262.693  2029.6 274.052  2036.6 289.044  2037.9 308.179  2035.7
 310.796 2038.39 321.634  2046.4 337.833 2057.53 344.024 2062.27
#Mann= 3 ,-1 , 0
       0     .05       0  178.03     .05       0 235.039     .05       0
#XS Ineff= 2 , 0
       0     160    2031     255       0    2031
Permanent Ineff=
       F       F
Bank Sta=178.03,235.039
Skew Angle= 15
Exp/Cntr=0.5,0.3

Type RM Length L Ch R = 3 ,10259   ,,,
Bridge Culvert--1,0,-1,-1, 0
Deck Dist Width WeirC Skew NumUp NumDn MinLoCord MaxHiCord MaxSubmerge Is_Ogee
15,12,2.6,15, 30, 39, , , 0.95, 0, 0,0,,
       0   6.462   8.519   9.225  17.522  18.353  27.703  27.954  36.406  41.313
  46.683   51.59  55.676  60.399  66.118  68.194  72.251  93.936 151.554 170.776
 238.777 243.413 285.045 289.642  290.27 299.485 303.117 303.407 304.131 338.074
 2036.49 2036.31 2036.25 2036.23 2035.87 2035.84 2035.37 2035.35 2034.79 2034.55
 2034.25 2033.97 2033.78 2033.51 2033.15  2032.4  2032.1  2031.1  2032.9  2032.9
  2032.9  2033.2  2037.4 2035.88 2035.85 2047.14  2051.6  2051.8 2052.27 2058.97
                                                                                
                                                                         2031.15
 2031.15
       0   6.462   8.519   9.225  17.522  18.353  27.703  27.954  36.406  41.313
  46.683   51.59  55.676  60.399  66.118  69.634   71.45  72.541  74.666  89.638
 123.445 191.446 201.202 223.254 263.601 267.281 268.238 269.049 269.831 276.689
  279.51 283.354 289.642  290.27 299.485 303.117 303.407 304.131 317.171
 2036.49 2036.31 2036.25 2036.23 2035.87 2035.84 2035.37 2035.35 2034.79 2034.55
 2034.25 2033.97 2033.78 2033.51 2033.15 2032.88  2032.7  2032.4  2032.1  2031.1
  2032.9  2032.9  2032.9  2033.2  2037.4 2037.57 2037.69 2037.74 2037.71 2037.03
 2036.81  2036.6 2035.88 2035.85 2047.14  2051.6  2051.8 2052.27 2058.97
                                                                                
                                                                                
 2031.15 2031.15
                                                                        
Pier Skew, UpSta & Num, DnSta & Num=  ,181.594, 4 ,141.025, 4 , 0 , 0 , 0 ,,
       3       3       2       2
    2020    2022    2022  2032.9
       3       3       2       2
    2020    2022    2022  2032.9
Pier Skew, UpSta & Num, DnSta & Num=  ,216.367, 2 ,170.003, 2 , 0 , 0 , 0 ,,
       2       2
    2031 2031.15
       2       2
    2031 2031.15
BR Coef=-1 , 0 , 0 ,, 0 ,,,0.8,0,,0,
WSPro=,,,, 1 ,,,, 0 ,,,, 0 ,,,,-1 ,-1 ,-1 , 0 , 0 , 0 , 0 , 0
BC Design=,, 0 ,, 0 ,,,,,,

Type RM Length L Ch R = 1 ,10244   ,66.96,74.79,84.65
XS GIS Cut Line= 6
  955016.1606273  766068.2008603  954944.3956352  766094.9108764
  954905.9004031  766087.0998044   954841.500019  766044.2996763
   954804.499827  766007.5001882  954735.6716669  765958.0389402
#Sta/Elev= 30
       0 2034.66  18.488 2035.05  28.302 2034.22  39.873 2033.99   43.67 2033.48
  43.882    2033 108.155  2029.6 117.176  2027.7 139.325    2025 145.362  2022.1
 148.637  2021.1 151.428  2020.5  156.47  2020.8 161.706  2020.1 169.317    2021
 188.771  2026.4 200.101  2030.2 209.055  2030.5 239.173  2029.7 240.071 2031.82
   243.8 2033.56 249.769 2034.63  259.38 2036.85 267.658 2037.04 282.031 2036.27
 288.966 2036.17  297.38 2045.82 306.247 2054.24 310.854 2057.36 321.035 2063.34
#Mann= 3 ,-1 , 0
       0     .05       0 148.637    .055       0 169.317     .05       0
#XS Ineff= 2 , 0
       0  104.96    2030  209.05       0    2030
Permanent Ineff=
       F       F
Bank Sta=148.637,169.317
Skew Angle= 15
Exp/Cntr=0.5,0.3

Type RM Length L Ch R = 1 ,10170   ,237.49,225.25,213.35
XS GIS Cut Line= 6
  955057.8998913  766096.7192604  955011.8188673  766044.2239003
  954959.1002752  766064.6998043  954922.2997631  766016.8001563
  954896.8226431  765948.6140442  954792.3306109  765883.2388121
#Sta/Elev= 30
       0 2040.31   20.65 2037.39   27.92 2035.85   59.32 2033.77   75.59 2031.48
  108.26 2030.66  126.41 2029.44  135.56 2028.13  146.61 2025.47  153.58  2025.2
  154.782023.182  155.84  2021.4   171.9  2020.9  186.46  2021.5  188.79  2023.1
  194.98 2027.14  225.21 2026.22  256.67    2026  287.45 2026.51  314.91 2027.98
  324.32 2029.47  331.59 2031.95  335.91  2034.4  338.21 2034.86  343.31 2037.21
  350.02 2036.87  357.76 2037.61  362.24 2037.06  368.88 2039.61  384.41 2051.25
#Mann= 3 ,-1 , 0
       0     .07       0  153.58    .055       0  188.79     .05       0
Bank Sta=154.78,188.79
Exp/Cntr=0.3,0.1

Type RM Length L Ch R = 1 ,9944    ,340.22,327.57,310.81
XS GIS Cut Line= 6
  955306.3693957  766120.5293084  955181.1690115  765916.2556441
  955110.5672834  765880.4842521  955024.9045633   765854.126492
  954908.1767551   765833.417116   954864.999795   765825.849756
#Sta/Elev= 30
       0  2061.5   12.29 2056.82    58.6 2050.89   88.97 2047.49  114.86  2043.4
  122.79 2041.69  160.47 2035.14  200.16 2031.79  242.98 2029.76  266.88 2028.76
  321.19 2028.07  335.74 2025.19  349.35  2022.2  354.89 2019.96  361.07 2021.62
  375.67 2022.52  382.64 2022.11  390.18 2027.71  395.98 2029.65  401.02 2029.38
  421.64  2026.6  460.92 2025.66  490.84 2025.46  529.19  2026.1  535.49 2027.05
  542.61  2027.5  546.72 2028.57  558.23 2034.45  564.19 2038.23  570.75 2038.96
#Mann= 5 ,-1 , 0
       0     .05       0  335.74     .07       0  349.35    .055       0
  361.07     .07       0  421.64     .05       0
Bank Sta=349.35,361.07
Exp/Cntr=0.3,0.1

Type RM Length L Ch R = 1 ,9617    ,342.67,347.34,346.61
XS GIS Cut Line= 6
  955702.5918602  765605.4614037   955542.649204  765507.7083155
  955351.5544197  765470.0537875  955270.5980036  765472.8779795
  955064.4412033  765539.7144596   954830.963059  765667.5465238
#Sta/Elev= 30
       0 2066.64   12.56 2061.69   57.88 2051.95   72.91 2049.97  118.07 2045.78
  247.81 2038.49  315.36 2035.41  399.03 2029.56  425.65 2028.56  496.58 2027.55
  586.65 2027.46  639.33 2026.58  683.71 2026.87  698.79 2022.19  705.52 2020.02
  713.63 2020.72     719 2022.52  724.59 2023.61  737.06 2023.82  753.05 2020.97
  763.06 2020.22  770.53 2024.48  785.23 2026.58  818.17 2024.63  843.87 2024.49
  911.79 2028.46  924.59 2030.46  938.37 2034.51  946.93 2038.04  948.42 2038.08
#Mann= 4 ,-1 , 0
       0     .05       0  586.65     .07       0  698.79     .05       0
     719     .05       0
#XS Ineff= 2 , 0
       0     550    2040               0
Permanent Ineff=
       F       F
Bank Sta=698.79,719
Exp/Cntr=0.3,0.1

Type RM Length L Ch R = 1 ,9270    ,353.71,355.41,362.7
XS GIS Cut Line= 2
  954962.3299712  765310.0394513  954617.0177147  765470.3630355
#Sta/Elev= 30
       0 2063.46   33.05 2054.65   39.47 2053.21    54.1 2049.17   64.03 2045.35
   90.11 2034.19   97.54 2030.11  114.77 2027.75  152.49 2023.03     165 2022.59
  176.96 2022.86   198.3 2023.79  209.53 2023.06  231.31 2019.67  233.04 2019.64
  238.84 2018.72  247.79 2018.16  255.62 2018.95  258.67  2019.5  268.36 2024.76
  275.47    2029  289.11 2032.55  304.42 2034.28  306.87 2034.29  313.12  2036.1
  332.46 2053.56  336.68 2057.82  355.88 2070.27  369.87  2080.9  380.72 2086.34
#Mann= 6 ,-1 , 0
       0     .08       0  114.77     .05       0  233.04     .05       0
  255.62     .05       0  275.47     .03       0  313.12     .05       0
Bank Sta=233.04,255.62
Exp/Cntr=0.3,0.1

Type RM Length L Ch R = 1 ,8914    ,50.8,51.82,45.69
XS GIS Cut Line= 6
  955031.0116993   765080.181147   954809.300339  765052.5997069
  954747.4998909  765057.8999309  954695.3997948  765065.2000269
  954651.0554747   765079.509403  954585.9382907   765127.843227
#Sta/Elev= 30
       0 2077.83   26.49 2073.65   54.68 2067.87   87.84 2060.58  101.62 2055.35
  117.58 2053.14  143.45 2048.08  165.28 2040.11  192.79 2033.44  213.96 2031.08
  223.42    2030     236  2025.3  275.06  2021.2  286.19  2014.3   288.8  2013.3
  303.34  2012.7  310.67  2013.7  319.88  2013.8  322.87  2015.2  332.54  2016.8
   347.5  2026.2  358.99  2027.7  377.92    2026  381.25 2027.65  385.26 2027.59
  401.47 2043.03   411.8  2056.2  420.35 2059.31   460.8 2077.85  467.31 2079.99
#Mann= 5 ,-1 , 0
       0     .07       0  117.58     .03       0  213.96     .07       0
  286.19    .055       0  310.67     .05       0
Bank Sta=286.19,310.67
Exp/Cntr=0.5,0.3

Type RM Length L Ch R = 1 ,8862    ,31.67,29.84,34.21
XS GIS Cut Line= 6
  955041.0817153  765052.6570509  954783.5999869  765003.3002508
  954703.5999868  765011.4000909  954681.1999868  765028.4998669
  954669.9001468  765032.1002509  954638.7265147  765050.9510669
#Sta/Elev= 30
       0 2078.23   20.64  2074.9   74.21 2062.61    97.4 2054.83  113.47 2051.95
  135.73 2048.77  144.89 2046.88  161.37 2041.03  184.31 2035.58  192.16 2033.82
  209.68 2030.66  228.38 2027.72  247.76 2025.29  261.72 2024.31  262.15  2023.6
  288.68  2021.7   304.3  2014.5  308.55    2013  325.22  2012.6  333.27  2013.1
  344.17  2013.5  345.14  2014.2   353.1  2016.6  359.67  2019.7  372.76  2020.9
  384.64  2026.9  392.44 2025.59  404.28 2027.24  415.09 2027.45  421.06 2032.62
#Mann= 5 ,-1 , 0
       0     .07       0  184.31     .03       0  228.38     .07       0
  308.55     .05       0  333.27     .05       0
#XS Ineff= 2 , 0
       0     290    2024     350       0    2024
Permanent Ineff=
       F       F
Bank Sta=308.55,333.27
Exp/Cntr=0.5,0.3

Type RM Length L Ch R = 3 ,8852    ,,,
Bridge Culvert--1,0,-1,-1, 0
Deck Dist Width WeirC Skew NumUp NumDn MinLoCord MaxHiCord MaxSubmerge Is_Ogee
10.5,12.9,2.6,0, 67, 66, , , 0.95, 0, 0,0,,
       0    1.15    7.71    8.25    8.78   16.37   18.78    23.5   31.07   32.45
   38.87      46   47.14   52.04   54.56   55.83   61.21   64.63   69.78   82.73
   84.72   86.91   93.12   98.38  102.25  112.67  115.98  116.46  128.74  144.89
  146.27   147.8  160.11  163.06  176.02   177.7  178.84   180.3   182.9  199.13
  203.24  208.27  210.68  214.48  219.53  224.39  226.88  229.92  229.99   230.9
   238.2   271.1   297.5   342.5   345.1   362.6   387.8  393.36  394.11  398.36
  402.69  407.77  415.47  417.43  418.69  427.58  431.05
 2077.97 2077.75 2076.06 2075.96 2075.84 2075.09 2074.47 2073.19 2071.65 2071.33
 2070.12    2068 2067.74  2066.5 2065.84 2065.55 2064.29 2063.45  2062.3 2058.07
 2057.46 2057.05  2055.7 2054.92 2054.24 2051.71 2050.82 2050.65 2048.28 2045.76
 2045.48 2044.91 2040.31 2039.54 2036.85 2036.47 2036.22 2035.87  2035.3 2031.32
 2030.44 2029.65 2029.26 2028.78 2028.27 2027.55 2027.26 2026.93 2026.92  2026.5
    2026  2024.3  2025.2  2025.2    2025  2025.4  2026.9 2026.87 2026.96 2027.42
 2027.57 2027.64 2027.67 2027.68 2027.56 2029.31    2031
                                                                                
                                                                                
                                                                                
                                                                                
                                                                                
                  2022.7  2022.7
                                                        
       0    1.15    7.71    8.25    8.78   16.37   18.78    23.5   31.07   32.45
   38.87      46   47.14   52.04   54.56   55.83   61.21   64.63   69.78   82.73
   84.72   86.91   93.12   98.38  102.25  112.67  115.98  116.46  128.74  144.89
  146.27   147.8  160.11  163.06  176.02   177.7  178.84   180.3   182.9  199.13
  203.24  208.27  210.68  214.48  219.53  224.39  226.88  229.92  229.99   230.9
   238.2   271.1   301.5   317.5   362.6   387.8  393.36  394.11  398.36  402.69
  407.77  415.47  417.43  418.69  427.58  431.05
 2077.97 2077.75 2076.06 2075.96 2075.84 2075.09 2074.47 2073.19 2071.65 2071.33
 2070.12    2068 2067.74  2066.5 2065.84 2065.55 2064.29 2063.45  2062.3 2058.07
 2057.46 2057.05  2055.7 2054.92 2054.24 2051.71 2050.82 2050.65 2048.28 2045.76
 2045.48 2044.91 2040.31 2039.54 2036.85 2036.47 2036.22 2035.87  2035.3 2031.32
 2030.44 2029.65 2029.26 2028.78 2028.27 2027.55 2027.26 2026.93 2026.92  2026.5
    2026  2024.3  2025.2    2025  2025.4  2026.9 2026.87 2026.96 2027.42 2027.57
 2027.64 2027.67 2027.68 2027.56 2029.31    2031
                                                                                
                                                                                
                                                                                
                                                                                
                                                                                
                          2022.5  2022.9
                                                
BR Coef=-1 , 0 , 0 ,, 0 ,,,0.8,0,,0,
WSPro=,,,, 1 ,,,, 0 ,,,, 0 ,,,,-1 ,-1 ,-1 , 0 , 0 , 0 , 0 , 0
BC Design=,, 0 ,, 0 ,,,,,,

Type RM Length L Ch R = 1 ,8832    ,36.09,33.93,29.94
XS GIS Cut Line= 6
  955044.5735553  765034.6745869   954808.599923  764970.1001228
  954749.1997309  764972.5003788  954665.0003068  764991.6000268
  954646.4996987  765000.5999628  954620.4163707  765032.1473549
#Sta/Elev= 30
       0 2078.15   16.05 2074.96   31.37 2071.26   38.27 2070.35   58.23  2064.3
   84.53 2057.24   92.69 2055.59   114.5 2050.16   126.7 2046.03  152.77 2039.32
  170.61 2037.72  208.09 2028.73  244.66  2024.9  304.09  2018.1  321.24    2014
  323.01  2013.8  324.58 2013.19   325.5  2012.6  351.43  2012.7  355.44 2013.25
   358.9  2013.7  378.37    2019  391.13  2019.6  398.87  2020.9  411.73  2027.2
  418.98 2027.19  429.59 2027.74     441 2027.08  443.71 2027.18  452.66 2031.76
#Mann= 3 ,-1 , 0
       0     .07       0  324.58     .05       0  355.44     .05       0
#XS Ineff= 2 , 0
       0     300    2022     380       0    2022
Permanent Ineff=
       F       F
Bank Sta=324.58,355.44
Exp/Cntr=0.5,0.3

Type RM Length L Ch R = 1 ,8799    ,281.91,254.58,231.82
XS GIS Cut Line= 6
   954815.369587  764887.6875787  954778.5997949  764924.8997387
  954720.2000508  764944.9998348  954686.2001788  764952.5999628
  954637.7997947  764977.8999308  954595.6150907  765018.7687949
#Sta/Elev= 25
       0 2034.47    1.69 2033.72   17.16 2029.38   18.02 2029.31   19.43 2028.97
   32.79 2026.26   44.08 2024.35   47.27 2023.89   52.33  2022.3  108.06  2015.1
  111.66 2013.75  114.78 2012.45  131.02 2012.45  148.93  2013.8  154.09  2015.7
  203.56  2019.4  223.47 2028.16  227.69 2028.24  232.51  2028.3  239.09 2028.24
  245.41 2027.81  249.44 2027.91  253.32 2030.05  259.88 2032.72  262.28 2033.89
#Mann= 3 ,-1 , 0
       0     .09       0  111.66     .05       0  148.93     .05       0
Bank Sta=111.66,148.93
Exp/Cntr=0.3,0.1

Type RM Length L Ch R = 1 ,8544    ,53.5,50.2,41.99
XS GIS Cut Line= 6
  954491.5326585  764762.0202505  954473.1999865  764803.5004426
  954473.3996665  764839.3998346  954467.8004345  764870.4004107
  954477.4004345  764935.8002188  954476.3876985  765010.7662349
#Sta/Elev= 30
       0 2055.69    6.97 2052.92   12.62  2050.8   23.42 2044.34   34.32    2038
   45.37  2037.1   67.68    2023   81.57  2011.6   83.12  2011.1   97.45  2010.5
  106.07  2010.6  113.15    2011  116.05  2011.5  118.39  2012.5  143.86  2018.3
  179.45  2020.4   181.6 2021.83   186.7 2022.02  191.25  2022.9  195.48 2024.31
  200.75 2026.34  204.58 2027.95  209.82  2028.8  216.83 2028.97  219.75 2029.05
  221.26 2029.04  232.96 2028.87  241.41 2034.45  246.65 2038.03  254.44 2042.16
#Mann= 4 ,-1 , 0
       0     .09       0   81.57    .055       0  116.05     .07       0
  143.86     .05       0
Bank Sta=81.57,116.05
Exp/Cntr=0.5,0.3

Type RM Length L Ch R = 1 ,8494    ,30.72,34.57,33.76
XS GIS Cut Line= 6
  954405.2514424  764749.6288265  954419.2003704  764854.4004106
  954430.6998904  764898.0996107  954431.2999544  764913.8999307
  954428.2996344  764919.3404427  954434.8788344  765008.6004749
#Sta/Elev= 25
       0 2036.34   13.04 2034.33   19.96 2032.66   24.75  2031.7   57.37  2026.8
    74.6  2020.5    80.7  2019.2   84.15  2014.7   93.04  2012.6   96.62  2011.2
   98.49  2010.8  106.27  2010.2  115.27    2010  122.16  2010.8     129  2011.8
  151.52  2017.3  167.33  2025.2  173.54 2025.93  205.44  2028.5  213.45 2029.47
  228.77 2029.68  233.91 2029.92  240.32 2030.08  258.53  2039.6  263.05 2042.09
#Mann= 3 ,-1 , 0
       0     .08       0   98.49    .055       0  122.16     .05       0
#XS Ineff= 2 , 0
       0   50.25    2027   178.5       0    2027
Permanent Ineff=
       F       F
Bank Sta=98.49,122.16
Exp/Cntr=0.5,0.3

Type RM Length L Ch R = 3 ,8479    ,,,
Bridge Culvert--1,0,-1,-1, 0
Deck Dist Width WeirC Skew NumUp NumDn MinLoCord MaxHiCord MaxSubmerge Is_Ogee
9.5,12,2.6,0, 19, 19, , , 0.95, 0, 0,0,,
       0    2.63    4.29   10.82   18.22   18.47   18.68   22.43   27.73      72
   151.9   159.9   183.1   214.3   225.9   235.7   241.7   245.4  251.42
 2035.82 2035.46 2035.23 2034.25  2033.3 2033.27 2033.24  2032.7  2032.2  2026.6
  2026.6  2026.6  2026.4  2029.4  2029.6  2028.8 2036.67 2038.75 2042.39
                                                                          2024.2
  2024.2
       0    2.63    4.29   10.82   18.22   18.47   18.68   22.43    25.8      76
   155.9   160.4   181.1   211.6   222.7   231.2   241.7   245.4  251.42
 2035.82 2035.46 2035.23 2034.25  2033.3 2033.27 2033.24  2032.7  2032.2  2026.6
  2026.6  2026.6  2026.4  2029.4  2029.6  2028.8 2036.67 2038.75 2042.39
                                                                          2024.2
  2024.2
Pier Skew, UpSta & Num, DnSta & Num=  ,85, 6 ,87, 6 , 0 , 0 , 0 ,,
       4       4       2       2      .5      .5
    2014    2016    2016  2023.2  2023.2  2024.2
       4       4       2       2      .5      .5
    2014    2016    2016  2023.2  2023.2  2024.2
Pier Skew, UpSta & Num, DnSta & Num=  ,109, 6 ,111, 6 , 0 , 0 , 0 ,,
       4       4       2       2      .5      .5
    2010    2012    2012  2023.2  2023.2  2024.2
       4       4       2       2      .5      .5
    2010    2012    2012  2023.2  2023.2  2024.2
Pier Skew, UpSta & Num, DnSta & Num=  ,134, 6 ,137, 6 , 0 , 0 , 0 ,,
       4       4       2       2      .5      .5
    2013    2015    2015  2023.2  2023.2  2024.2
       4       4       2       2      .5      .5
    2013    2015    2015  2023.2  2023.2  2024.2
BR Coef=-1 , 1 , 0 ,, 0 ,,,0.8,0,2,0,
WSPro=,,,, 1 ,,,, 0 ,,,, 0 ,,,,-1 ,-1 ,-1 , 0 , 0 , 0 , 0 , 0
BC Design=,, 0 ,, 0 ,,,,,,

Type RM Length L Ch R = 1 ,8459    ,60.29,52.6,55.65
XS GIS Cut Line= 6
  954366.5923704  764754.5645065  954368.9004664  764780.5997065
  954389.2002424  764841.6004106  954386.0995704  764870.4997387
  954394.8998264  764887.8995467  954399.2589944  765005.4895628
#Sta/Elev= 28
       0 2037.09     1.9 2036.73    10.2 2035.45   14.13 2035.07   19.46 2034.22
   24.21  2033.7   26.13    2033   44.86  2031.6   57.18  2029.2   78.28  2016.5
   90.46  2013.3   95.03  2012.5   96.42  2011.1   99.87  2010.3  105.59  2009.8
  119.71  2010.4   129.5  2010.5  135.66  2011.1  139.88  2012.8  154.98  2016.8
   205.9  2029.4  216.27 2029.93   220.7 2029.76  230.49 2029.44  235.77 2032.37
  245.86    2038  252.86 2040.71  257.66 2043.71
#Mann= 3 ,-1 , 0
       0     .07       0   96.42     .05       0  135.66     .05       0
#XS Ineff= 2 , 0
       0    63.2  2026.2     178       0  2026.2
Permanent Ineff=
       F       F
Bank Sta=96.42,135.66
Exp/Cntr=0.5,0.3

Type RM Length L Ch R = 1 ,8407    ,161.99,160.34,158.32
XS GIS Cut Line= 6
  954319.4330743  764776.4924425  954330.7001463  764828.7000586
  954328.4995703  764853.3999626  954340.7998583  764907.6002827
  954356.7998583  764953.3997068  954357.3302903  765003.8767628
#Sta/Elev= 28
       0 2039.82   10.05 2035.47   11.72 2034.92   13.76 2034.37   21.91  2032.8
   24.05  2039.3   41.98  2030.4   53.53  2024.3   66.05  2014.1   78.34  2010.5
   86.86  2009.9  102.41  2009.5  114.43  2009.7  118.93  2010.5  121.75  2010.9
  134.18  2016.3  152.96  2016.9  163.92  2018.5  182.76  2029.6  188.21 2030.02
  196.16 2030.59  198.26 2030.64   212.1 2031.17  212.69 2031.18   212.9 2031.32
  220.78 2036.95  227.74 2040.47  233.24  2043.5
#Mann= 3 ,-1 , 0
       0     .08       0   78.34     .05       0  118.93     .05       0
Bank Sta=78.34,118.93
Exp/Cntr=0.3,0.1

Type RM Length L Ch R = 1 ,8246    ,366.36,360.51,348.69
XS GIS Cut Line= 4
  954161.1533941  764845.2448266  954176.2717301  764897.5302667
  954187.6104821  764947.9254028  954233.5962742  765020.9990669
#Sta/Elev= 28
       0  2041.4    9.53 2038.66   16.93 2036.15   29.26 2023.39   37.18 2017.54
   41.96 2015.47   59.32 2010.63   66.75 2010.22   72.39 2009.41   73.12 2009.43
   80.05 2010.21   85.85 2010.45   99.29 2012.39  108.02  2014.1  110.48 2014.36
  122.72 2016.15   126.6 2016.55  129.26 2017.03  136.33 2017.91  142.75 2019.34
  154.39  2026.7  161.34 2030.25  165.99 2031.53  170.73 2031.36  174.58 2031.46
  183.81 2031.08  186.46 2031.15  192.42 2031.68
#Mann= 3 , 0 , 0
       0      .1       0   66.75    .055       0   80.05     .07       0
Bank Sta=66.75,80.05
Exp/Cntr=0.3,0.1

Type RM Length L Ch R = 1 ,7886    ,355.61,356.83,362.71
XS GIS Cut Line= 4
  953840.6895216  765034.5619469  953889.9039857   765119.210907
  953912.5425777   765144.802715  953972.5837938  765191.0639631
#Sta/Elev= 26
       0  2064.9    8.43 2060.84   16.81 2056.04   24.54 2051.81   30.78 2049.42
   49.89 2039.47   53.93 2036.71   75.78 2024.99   78.88 2023.08    93.8 2010.77
   98.06 2007.45   99.02 2006.73   105.9 2006.93  114.69 2007.16  118.65 2007.12
  129.52  2007.3  132.09 2007.51  154.76 2012.24  160.13 2012.54  163.96 2013.31
  167.83 2013.99  168.53 2014.05   189.8  2021.6   195.6 2022.74  202.06 2023.72
  207.89  2024.3
#Mann= 3 , 0 , 0
       0      .1       0   98.06    .055       0   105.9     .07       0
Bank Sta=98.06,105.9
Exp/Cntr=0.3,0.1

Type RM Length L Ch R = 1 ,7529    ,68.59,67.07,67.96
XS GIS Cut Line= 6
  953553.5619692  765237.4634512  953586.4999533  765303.0004753
  953595.9996013  765312.0997393  953604.9995373  765328.0997393
  953607.3997933  765344.0997393  953669.6784494  765420.8137234
#Sta/Elev= 30
       0 2021.46     .82 2021.08    8.18  2018.3     9.4 2017.97   19.29 2016.85
   33.12 2015.65   38.64  2015.3    44.9 2014.56   47.59 2014.12    60.8 2010.91
   66.69 2009.18   70.26 2008.51   73.35  2006.3      80  2005.3   81.98  2002.9
   83.79  2002.7   86.54  2002.1   96.69  2001.5  104.93  2002.1  107.22  2002.5
  108.94  2003.5  121.27  2008.8  155.33  2011.1  181.45  2015.4  198.96  2017.9
  201.66 2018.53  206.62 2018.64  209.33  2018.6  216.28 2019.26  220.26 2020.05
#Mann= 3 ,-1 , 0
       0     .05       0   86.54     .05       0  104.93     .05       0
Bank Sta=86.54,104.93
Exp/Cntr=0.5,0.3

Type RM Length L Ch R = 1 ,7462    ,44.89,49.53,43.58
XS GIS Cut Line= 6
  953479.1724651  765254.8079632  953527.3997932  765335.9998993
  953537.1001452  765344.0997393  953541.5002732  765364.3995153
  953579.9996013  765420.2003474  953621.2115053  765473.3735955
#Sta/Elev= 30
       0  2024.1    1.72 2023.64    3.48 2022.84   17.95 2017.73   19.93 2017.64
   24.79    2016   60.68  2010.8   77.62  2006.7   85.64  2003.7   90.57  2002.2
    97.7 2001.12  102.63  2000.3  111.48  1999.8  113.272000.681  116.15  2002.1
   117.3  2003.3  140.76  2008.6  179.36  2013.6  180.47  2012.3  185.02 2012.68
   190.3 2013.62  199.93  2014.9  202.76 2015.13  219.47 2017.07  222.23  2017.3
  236.28 2018.05  243.96 2018.29  248.82  2017.8  260.63 2025.47   263.7  2027.7
#Mann= 3 , 0 , 0
       0     .05       0    97.7     .05       0  113.27     .05       0
#XS Ineff= 2 , 0
       0      70 2012.65     150       0 2012.65
Permanent Ineff=
       F       F
Bank Sta=97.7,113.27
Exp/Cntr=0.5,0.3

Type RM Length L Ch R = 3 ,7444    ,,,
Bridge Culvert--1,0,-1,-1, 0
Deck Dist Width WeirC Skew NumUp NumDn MinLoCord MaxHiCord MaxSubmerge Is_Ogee
11,12,2.6,0, 27, 28, , , 0.95, 0, 0,0,,
       0     .05    1.22    3.34   24.62    64.9      80     137   156.7   195.8
  198.23  204.04  206.73  212.21  214.37  220.24  222.08  226.29   229.8     236
  238.75  241.99  246.29  251.87  255.47  258.91  274.23
 2021.97 2021.96 2021.59  2015.2  2015.2  2014.3  2013.2  2013.2  2013.5  2014.7
 2014.04 2014.46 2014.75 2015.22  2015.4 2015.81 2015.94 2016.29 2016.68 2017.19
 2017.34 2017.54 2017.88 2018.08 2018.19 2018.39 2029.58
                                                  2011.7  2011.7
                                                                                
                                                        
       0     .05    1.22   12.21    13.7   33.67    66.9      75     135   153.8
     194  198.23  204.04  206.73  212.21  214.37  220.24  222.08  226.29   229.8
     236  238.75  241.99  246.29  251.87  255.47  258.91  274.23
 2021.97 2021.96 2021.59 2019.21  2015.2  2015.2  2014.3  2013.2  2013.2  2013.5
  2014.7 2014.04 2014.46 2014.75 2015.22  2015.4 2015.81 2015.94 2016.29 2016.68
 2017.19 2017.34 2017.54 2017.88 2018.08 2018.19 2018.39 2029.58
                                                          2011.7  2011.7
                                                                                
                                                                
BR Coef=-1 , 0 , 0 ,, 0 ,,,0.8,0,,0,
WSPro=,,,, 1 ,,,, 0 ,,,, 0 ,,,,-1 ,-1 ,-1 , 0 , 0 , 0 , 0 , 0
BC Design=,, 0 ,, 0 ,,,,,,

Type RM Length L Ch R = 1 ,7412    ,43.59,41.12,39.76
XS GIS Cut Line= 6
  953440.0106091  765263.9870992  953477.5002731  765322.5998353
  953493.3999211  765369.2000274  953524.0001132  765417.6004114
  953540.1997932  765451.1998995  953584.6127213  765500.2372115
#Sta/Elev= 28
       0 2022.19   11.75  2019.3   13.91 2018.93    21.4 2017.99   25.61 2016.51
   29.62 2016.09   36.04 2015.96   37.91  2011.7   55.03    2010   76.96  2005.2
   84.36  2002.2   87.22  2001.1   96.18 1999.75  107.81  2001.1  109.74  2002.2
  115.76  2004.8  133.61  2010.4  145.12  2010.3   182.4  2012.2  188.52 2012.55
  196.13 2013.13  202.22 2013.38   220.3  2014.9  246.25 2017.43  262.27 2018.37
  268.72 2019.63  270.12 2019.77  280.24 2027.83
#Mann= 4 ,-1 , 0
       0     .05       0   25.61     .03       0   84.36     .05       0
  109.74     .05       0
#XS Ineff= 2 , 0
       0      70    2011     150       0    2011
Permanent Ineff=
       F       F
Bank Sta=84.36,109.74
Exp/Cntr=0.5,0.3

Type RM Length L Ch R = 1 ,7371    ,219.74,225.71,235.91
XS GIS Cut Line= 6
   953392.281969  765284.1803792  953449.1999851  765376.3004434
  953484.0999531  765426.8000274  953507.1000171  765466.2004755
  953527.4796652  765494.2601235  953554.1763692  765521.2742676
#Sta/Elev= 27
       0 2021.98    5.75 2021.18    8.92 2020.66   19.09  2017.5   22.59    2012
   46.29  2010.9   75.33  2006.9   79.27  2005.3   83.37  2004.6   87.96    2002
   89.36  2001.2  101.48  1999.7  114.36  2001.3  116.85  2002.1  117.39  2003.1
  141.04  2009.9  150.74  2009.8  186.66  2012.3  221.33 2016.65   223.6 2014.13
  235.44 2014.71  245.31 2015.73  257.54 2017.33  259.34 2017.48  264.91 2017.76
  275.99 2018.09  288.42 2025.32
#Mann= 3 ,-1 , 0
       0     .05       0   87.96     .05       0  116.85     .05       0
#XS Ineff= 2 , 0
       0                  221.33       0  2016.8
Permanent Ineff=
       F       F
Bank Sta=87.96,116.85
Exp/Cntr=0.3,0.1

Type RM Length L Ch R = 1 ,7145    ,325.66,369.19,412.3
XS GIS Cut Line= 6
  953260.7553128  765333.3180433  953241.3740648  765398.9175314
  953241.3740648  765438.4254995  953248.8287848  765477.9344915
  953260.0108648  765513.7150996  953277.9011688  765593.4775317
#Sta/Elev= 30
       0 2022.06    3.98 2021.85   11.52 2020.77   18.26 2019.51   31.01 2016.61
   44.99 2013.94   68.41  2007.6   73.38 2006.37   83.49 2006.51   88.59 2006.33
  107.91 2003.94  120.45 2002.55  123.11 2001.64  128.41 1999.61  131.35 1999.61
  136.47 2001.73  138.71 2002.51  149.45 2004.27  162.68 2009.26  167.43 2009.74
  179.91 2009.94  198.23 2011.58  216.27 2012.42  223.41 2012.99  227.61 2014.06
  233.38 2014.72  243.47 2017.69  256.49 2024.28  259.53 2026.19  267.35 2031.75
#Mann= 3 ,-1 , 0
       0     .07       0  123.11     .05       0  136.47     .05       0
Bank Sta=123.11,136.47
Exp/Cntr=0.3,0.1

Type RM Length L Ch R = 1 ,6776    ,277,284.11,292.78
XS GIS Cut Line= 6
  953289.8276968  765263.2467472  953213.0471527  765248.3383312
  953167.5754087  765236.4107792  953121.3581926  765217.0295311
  953096.0131686  765219.2659471  952884.4496483  765246.8709392
#Sta/Elev= 30
       0 2024.13    4.25 2023.98    14.1 2021.15   40.79  2014.4   64.55 2011.06
   78.21 2008.47   87.17 2006.41  102.01 2000.27  125.22 1999.92  155.07 1999.51
  160.98 1999.91  166.38 2000.45  197.33 2005.99  208.81 2006.06  223.08 2006.42
  241.35 2006.18  267.97 2006.44  295.15 2007.84  313.42 2009.44  327.09 2010.15
  352.93  2009.6  363.82    2010  375.63 2008.82  383.36 2010.15  386.36 2010.28
  397.28 2012.88  400.25 2012.51  411.48 2016.91  412.65 2016.77  414.14 2017.19
#Mann= 5 ,-1 , 0
       0     .05       0   78.21     .07       0  125.22     .05       0
  160.98     .07       0  208.81     .05       0
#XS Ineff= 2 , 0
       0                     300       0    2016
Permanent Ineff=
       F       F
Bank Sta=125.22,160.98
Exp/Cntr=0.3,0.1

Type RM Length L Ch R = 1 ,6492    ,322.38,306.84,294.23
XS GIS Cut Line= 6
  953450.8435051  765200.6301711   953364.371825   765082.849691
  953327.1002729  765026.1968909  953289.8276968  764976.2523148
  953278.6466408  764957.6155148  953189.9385447  764909.1618827
#Sta/Elev= 30
       0 2026.18   17.13 2022.47   21.18 2020.54    46.9 2014.21   81.27 2008.17
   98.87 2005.83  105.12  2005.4  124.64 2005.31  133.99 2004.88   144.5 2004.23
  152.22 2003.26  176.18 2002.81  202.32 2001.83  227.97 1997.63  230.61 1997.51
  241.97  1997.1  250.42 1997.36  251.84  1997.8  269.12 2002.81  278.87 2010.48
   286.2 2010.01  295.29 2010.54  303.58 2014.68  314.99 2018.71  320.17 2021.75
  346.45  2039.6  378.51 2057.98  383.76 2060.58   392.8 2067.17  399.05 2070.24
#Mann= 4 ,-1 , 0
       0    .055       0  152.22     .07       0  230.61     .05       0
  251.84     .07       0
Bank Sta=230.61,251.84
Exp/Cntr=0.3,0.1

Type RM Length L Ch R = 1 ,6185    ,328.6,320.05,311.24
XS GIS Cut Line= 6
  953717.7112174  764842.0724746  953547.0052972  764803.3089546
  953501.5335531  764792.1278985  953455.3163371  764789.8914825
   953394.935153  764780.2003465  953280.1375848  764776.4740105
#Sta/Elev= 30
       0 2078.22     6.8 2077.89   20.35 2072.66   86.47 2039.69   94.43 2035.08
  106.87 2029.08  127.75 2020.22  137.02 2015.35  142.86 2011.43  176.27 1995.76
  192.14  1994.8  199.16 1994.25  213.55 1995.82  236.97 1999.54  268.21 2000.66
  275.54 2002.58  282.89 2007.87   289.8 2010.16   305.7 2011.62   328.1 2009.62
  331.47 2010.89  336.06 2011.61  346.74 2017.93  355.45 2024.54  366.82 2029.13
  381.97 2032.69  404.41  2042.3   415.1 2045.55  424.04 2047.51  444.16 2054.27
#Mann= 3 ,-1 , 0
       0      .1       0  192.14    .055       0  213.55     .05       0
Bank Sta=192.14,213.55
Exp/Cntr=0.3,0.1

Type RM Length L Ch R = 1 ,5865    ,423.04,420.03,416.86
XS GIS Cut Line= 5
  953658.8220014  764465.6244741  953467.9883371  764485.7511941
  953438.9159531  764493.9513861   953411.334513  764501.4050821
  953259.2653928  764550.6041862
#Sta/Elev= 30
       0 2118.79    8.47    2115   20.47 2108.87   29.65 2103.61   44.16 2094.41
   53.62 2089.12   59.67  2085.2   72.42 2075.74   76.95 2073.74   86.77 2066.82
  107.06 2054.08  113.93 2051.18  122.26 2045.74  147.57 2024.61  193.68  1991.7
  202.41 1991.26  213.03 1991.86  246.01 1995.29  258.74 1997.19  267.03 1997.49
  274.46  1998.4  303.66  2004.5  307.89  2006.4   319.7 2008.85  327.09 2011.06
  338.06 2011.32  370.95 2027.33  381.25 2030.62  391.74 2035.35  410.49 2041.89
#Mann= 3 ,-1 , 0
       0      .1       0  193.68    .055       0  213.03     .07       0
Bank Sta=193.68,213.03
Exp/Cntr=0.3,0.1

Type RM Length L Ch R = 1 ,5445    ,371.53,354.25,337.71
XS GIS Cut Line= 4
  953506.0063851  763981.0871294  953289.8276968  764105.5758336
  953238.3921768  764130.1753856  953095.2676966  764277.7726978
#Sta/Elev= 30
       0 2133.09    8.48 2128.52   34.92 2117.17   59.83 2104.04   70.13 2099.12
   75.78 2095.82   89.07 2086.28   97.96 2077.85  126.68 2065.33   172.4 2037.71
  182.21 2030.04  211.15    2016  224.33 2006.75  254.86 1989.02  271.09 1988.89
  281.79 1988.29   288.9 1989.06  299.69  1989.3  327.01 1993.29  339.99  1994.2
  378.76  1995.6  424.86  1999.6  434.17 2001.72   455.4 2010.14  470.59 2008.35
  482.13 2014.65  489.06  2017.5  492.08 2019.24  504.64 2023.02  512.08 2024.74
#Mann= 4 ,-1 , 0
       0      .1       0  271.09    .055       0   288.9     .07       0
  424.86     .05       0
Bank Sta=271.09,288.9
Exp/Cntr=0.3,0.1

Type RM Length L Ch R = 1 ,5091    ,428.71,443.76,454.07
XS GIS Cut Line= 4
  952934.2518883  763801.4355452  952925.3072483  764022.8315135
  952915.6161123  764118.9943296  952919.3434723  764244.9739778
#Sta/Elev= 30
       0 2050.56   10.55 2048.53   26.15 2044.25   38.81 2041.54   77.21  2031.3
   82.67 2029.29   96.79 2026.24  126.07 2016.31  152.17 2010.23  162.46 2007.01
  163.55 2007.08  169.47 2004.89  209.66 1992.35  223.85 1987.52  231.24 1986.72
  235.61 1985.82  244.18 1985.78  249.82 1985.67  255.63  1985.8  263.22 1986.33
  294.76 1991.62  318.33 1993.13  336.95 1996.26  358.15 2000.78  367.58 2003.78
  396.37 2006.03  415.18 2014.41  433.28 2020.81  436.47 2021.27  444.26 2025.45
#Mann= 4 ,-1 , 0
       0      .1       0  244.18    .055       0  255.63     .07       0
  367.58     .05       0
Bank Sta=244.18,255.63
Exp/Cntr=0.3,0.1

Type RM Length L Ch R = 1 ,4647    ,327.72,325.76,324.73
XS GIS Cut Line= 4
   952712.110448   763682.910617  952556.3129438  763884.1798653
  952495.9327837  763946.0519934  952418.4067676  764102.5939456
#Sta/Elev= 30
       0 2114.35   44.26 2096.17  107.69 2068.16  122.01 2060.53  136.71 2053.67
  154.61 2048.45   166.5 2043.36  195.17 2029.38  214.48  2014.2  246.47 1995.46
  256.06 1992.15  280.91 1990.03  286.17 1988.02  310.29 1983.09  316.94 1982.17
  329.25 1983.03  344.15 1984.88   355.5 1993.03   369.8 1997.77  377.13  2001.9
  387.13 2009.07  397.88 2017.64  407.91 2024.17  412.03 2025.34  422.04 2026.46
  440.66  2026.5  450.03 2025.73  452.18 2025.59  491.71 2046.09  515.67 2054.45
#Mann= 5 ,-1 , 0
       0      .1       0  310.29    .055       0  329.25     .07       0
  412.03     .03       0  450.03     .05       0
Bank Sta=310.29,329.25
Exp/Cntr=0.3,0.1

Type RM Length L Ch R = 1 ,4321    ,348.85,352.68,353
XS GIS Cut Line= 2
  952344.0315995  763623.3250809  952194.1435993  763802.6213372
#Sta/Elev= 26
       0 2035.53   43.72 2018.55   52.81  2014.6   69.91 2007.65   101.9 1989.58
  102.64 1989.28  111.34 1986.64  122.35 1982.72  132.67 1981.41  134.16 1981.14
   137.4 1980.81  145.09 1979.89  148.43 1981.04  162.85 1982.07  171.56 1985.28
  178.68 1987.01  181.07 1987.16  189.84 1988.37  194.19 1988.01  200.12 1990.16
   203.8 1991.95  225.65 2006.19  226.18  2006.4  226.99 2006.86  231.26 2008.56
   233.7  2009.2
#Mann= 3 ,-1 , 0
       0      .1       0   137.4    .055       0  148.43     .05       0
Bank Sta=137.4,148.43
Exp/Cntr=0.3,0.1

Type RM Length L Ch R = 1 ,3969    ,167.76,118.14,69.87
XS GIS Cut Line= 6
  952127.3542232  763409.9849206  952058.5997911  763440.8001527
   951980.200303  763509.5003128   951959.999855  763533.4004728
   951954.199919  763542.4004088  951943.9926831  763552.3074017
#Sta/Elev= 29
       0 2035.75    5.31 2032.68   10.78 2029.68   17.76 2027.72   20.56 2026.84
    27.8 2025.18   31.04 2024.39   40.22 2023.38    43.4 2022.53   50.43 2017.42
   54.37 2014.91    62.5  2015.3    62.7 2015.35   62.91  2015.3   75.36    2012
   94.41  2009.7  112.61  2005.8  115.14  2004.1   126.3  2003.6  153.92  1982.8
  164.31  1979.2  165.77  1978.3  169.24  1978.2  179.84  1977.5  194.13  1977.7
  202.84  1978.6  211.15  1983.7  221.87  1986.2  236.08  1995.8
#Mann= 4 ,-1 , 0
       0     .05       0   126.3     .07       0  169.24    .055       0
  202.84     .07       0
Bank Sta=169.24,202.84
Exp/Cntr=0.5,0.3

Type RM Length L Ch R = 1 ,3851    ,90.16,108.79,113.65
XS GIS Cut Line= 6
  951804.3293268  763228.9406964  951826.9003348  763328.0997365
  951849.9997268  763374.8002806  951864.8999509  763413.2996086
  951888.0003669  763452.4000247  951911.8217967   763503.127793
#Sta/Elev= 30
       0 1999.52    .643  1999.4   2.284  1998.5   8.773 1997.99   10.16 1996.93
  16.749  1996.5  24.797 1995.82  26.002 1995.86  28.585  1995.6  36.606 1995.83
  40.412 1995.73  45.551 1995.44  49.938 1995.43  55.511 1994.88  61.819 1995.03
  67.059  1993.3  93.647  1992.8 114.379  1980.8 120.055  1977.9 127.579  1977.3
 144.442  1977.9 164.903    1977 171.416 1977.97 176.189  1978.5 181.273  1980.3
 225.292    1992 241.095  1995.2 258.147  1997.1  261.26  1997.3 268.875  1997.6
#Mann= 4 ,-1 , 0
       0     .05       0  93.647     .07       0 144.442    .052       0
 171.416     .06       0
#XS Ineff= 2 , 0
       0   89.55  1997.6  253.22       0  1997.6
Permanent Ineff=
       F       F
Bank Sta=144.442,171.416
Skew Angle= 25
Exp/Cntr=0.5,0.3

Type RM Length L Ch R = 3 ,3800    ,,,
Bridge Culvert--1,0,-1,-1, 0
Deck Dist Width WeirC Skew NumUp NumDn MinLoCord MaxHiCord MaxSubmerge Is_Ogee
28,24.6,2.6,25, 20, 19, , , 0.95, 0, 0,0,,
       0   4.359   5.429   8.048  13.232  15.317  22.766  24.371  33.497  35.292
  41.953  44.228  50.209 124.617 225.127 238.631 296.272 296.399  298.13 303.903
 1992.95 1992.97    1993 1992.98 1993.09  1993.1 1993.34 1993.39 1993.42 1993.47
 1993.67 1993.72 1993.72 1993.72  1997.1  1997.7  1998.8 1999.07 1999.11 1999.23
                                                                                
                         1991.52  1994.9
       0   4.359   5.429   8.048  13.232  15.317  22.766  24.371  33.497  35.292
  41.953  44.228  53.409 153.918 185.159  219.78 236.456 259.838 311.217
 1992.95 1992.97    1993 1992.98 1993.09  1993.1 1993.34 1993.39 1993.42 1993.47
 1993.67 1993.72 1993.82  1995.3  1996.1  1996.8  1997.1  1997.7  1998.8
                                                                                
                  1991.6  1993.1
Pier Skew, UpSta & Num, DnSta & Num=  ,153.166, 2 ,81.568, 2 , 0 , 0 , 0 ,,
     2.2     2.2
    1992  1994.9
     2.2     2.2
    1992  1994.9
Pier Skew, UpSta & Num, DnSta & Num=  ,185.793, 2 ,114.195, 2 , 0 , 0 , 0 ,,
     2.2     2.2
    1992  1994.9
     2.2     2.2
    1992  1994.9
BR Coef=-1 , 0 , 0 ,, 0 ,,,0.8,-1,,0,
WSPro=,,,, 1 ,,,, 0 ,,,, 0 ,,,,-1 ,-1 ,-1 , 0 , 0 , 0 , 0 , 0
BC Design=,, 0 ,, 0 ,,,,,,

Type RM Length L Ch R = 1 ,3742    ,41.06,26.35,33.54
XS GIS Cut Line= 6
  951741.1249747  763278.5934324  951746.7999827  763315.1000565
  951774.5002067  763371.3995766  951780.6001747  763400.8999926
  951815.9998548  763473.4002167  951880.9941589  763589.5894009
#Sta/Elev= 30
       0 2014.63   2.628 2015.16   3.707 2014.97   14.61 2008.85  22.495 2006.35
  28.784 2002.97   33.47  2010.1    56.3  1988.5  71.879  1985.6  90.359    1980
  93.667  1977.4   98.55  1974.3 109.219  1976.4 110.778  1977.2 115.681  1979.7
 118.146  1977.4 140.469    1977 146.061  1977.7 155.867  1981.9 191.494  1982.6
 193.977 1983.61 196.687 1983.73 210.653 1985.34 214.695 1986.14 240.317 1993.09
 261.542 1994.42 283.004 1997.03 286.058 1998.25 294.052 1999.74 312.232 2000.11
#Mann= 3 ,-1 , 0
       0     .06       0  93.667    .056       0 110.778    .055       0
#XS Ineff= 2 , 0
       0   38.89  1993.9     168       0  1993.9
Permanent Ineff=
       F       F
Bank Sta=93.667,110.778
Skew Angle= 25
Exp/Cntr=0.5,0.3

Type RM Length L Ch R = 1 ,3716    ,377.28,360.59,347.99
XS GIS Cut Line= 6
  951689.0166866  763292.3273205  951711.4996306  763344.9005045
  951784.1002067  763463.9998967  951827.7000788  763515.3002488
  951832.7002708  763542.6000888  951864.0459349  763593.2430329
#Sta/Elev= 30
       0 2039.41     .44 2039.41   23.81 2028.74   31.58 2025.93      36 2024.69
   39.98 2020.59   45.17  2019.2   57.47  2011.3   80.81  1985.9   94.39  1979.9
   98.09    1977  109.55  1976.8   125.1    1977   130.1 1974.07   143.4  1975.9
  155.17  1979.1  197.87  1982.2  265.18  1989.9  284.22  1989.9  293.03  1986.1
   297.3 1987.67  300.72 1987.79   308.2 1989.08  314.72 1989.19   320.2 1989.77
  327.11 1991.73  333.87 1994.02  336.65 1994.58  349.25 2000.19  352.59 2000.34
#Mann= 3 ,-1 , 0
       0     .07       0   125.1     .04       0   143.4     .05       0
Bank Sta=125.1,143.4
Exp/Cntr=0.3,0.1

Type RM Length L Ch R = 1 ,3355    ,401.13,411.81,427.86
XS GIS Cut Line= 4
  951515.2787024   763678.259609  951620.0533585  763729.6193531
  951694.0127826  763772.7625211  952057.6433751  763957.6590334
#Sta/Elev= 30
       0 2058.82    4.35 2059.31   24.83 2048.96   38.84 2036.08   66.08 2012.24
   80.99 1998.16    97.6 1985.69  109.95 1980.15  116.06 1979.11  122.17 1976.73
  129.78 1975.25  142.76 1974.48  147.68 1974.76  154.96 1976.39  168.59 1979.07
  178.58 1982.35  190.87 1983.81  242.48 1986.66  299.94  1988.5  336.12 1989.05
  372.99 1988.88  429.93 1990.55  534.13 1996.57  539.93 1997.26  554.43 2001.14
  563.35 2004.48  568.19 2004.59  586.55 2007.02  600.92 2009.56  610.25 2012.45
#Mann= 3 , 0 , 0
       0     .07       0  122.17     .05       0  154.96     .05       0
#XS Ineff= 2 , 0
       0                     200       0    2020
Permanent Ineff=
       F       F
Bank Sta=122.17,154.96
Exp/Cntr=0.3,0.1

Type RM Length L Ch R = 1 ,2943    ,442.21,461.38,481.79
XS GIS Cut Line= 4
  951536.6301264  763971.6980734  951532.4460624  764081.5323136
  951532.4460624  764129.6500736  951618.2203985  764278.1884418
#Sta/Elev= 30
       0 1994.21   23.58 1991.78   35.38 1990.47    51.3 1987.56   57.19 1985.71
   68.56 1983.29    77.3 1981.71   89.45 1980.53   92.12 1980.11  106.86 1978.26
  118.83 1975.67  119.54 1975.41  122.07 1975.17  136.01 1973.72  138.65 1973.71
  147.33 1975.73  158.03 1977.93  162.56  1978.1  169.45 1979.74  182.23 1983.01
  185.96 1984.32  197.35 1985.68  199.71 1986.87  210.95  1995.1  216.62 1999.44
  218.16 2000.19  275.62  2043.7  311.73 2070.38  314.02  2071.9  329.56 2080.07
#Mann= 4 ,-1 , 0
       0     .08       0  122.07     .05       0  147.33     .05       0
  169.45     .08       0
Bank Sta=122.07,147.33
Exp/Cntr=0.3,0.1

Type RM Length L Ch R = 1 ,2482    ,355.34,369.95,381.45
XS GIS Cut Line= 5
  951491.6499023   763694.498201  951409.0131022   763707.050393
  951330.5593421   763711.234457   951284.533614  763723.7866491
  951157.9631179  763831.5288572
#Sta/Elev= 30
       0 2054.15    4.12 2053.19   41.27 2038.43   53.66 2032.89   81.07 2019.79
   84.94 2018.37   89.35  2015.8   95.64 2013.79  107.59 2007.43  125.01 2000.12
  150.96 1986.87  164.29 1978.28   173.2 1971.88  185.23 1970.41  186.28 1969.98
  192.89 1970.41  196.28  1970.6  203.25 1971.76     219 1977.12  228.34 1979.47
  233.99 1981.44  257.49 1993.77  267.18  2000.8  296.83 2019.36  315.16 2030.21
  330.07 2040.26  344.37 2050.22  355.83 2059.03  363.44 2063.45  376.07 2074.45
#Mann= 3 ,-1 , 0
       0     .09       0  185.23     .05       0  192.89     .05       0
Bank Sta=185.23,192.89
Exp/Cntr=0.3,0.1

Type RM Length L Ch R = 1 ,2112    ,233.9,233.73,231.88
XS GIS Cut Line= 4
  951542.9062224  763483.1978487  951427.8413902  763414.1587446
  951374.4930382  763391.1463926   951240.599918  763379.6397046
#Sta/Elev= 30
       0 2055.75    9.92 2052.87   24.33 2044.35   31.59 2039.41   54.22 2022.53
   70.76  2009.9   95.97 1990.24  118.14  1975.7  139.58 1969.56  147.29 1968.39
  153.99 1967.94  157.05 1968.02  161.19 1967.61  167.76 1968.17  173.16 1967.94
  177.54 1968.19  181.58  1968.8  188.99 1971.92  211.15 1973.06  219.05 1972.81
  232.01 1974.96  234.36 1975.65  241.77 1979.63  260.47 1988.52  264.41 1989.56
  279.99    1993  299.19 1999.23  304.86 2002.74  310.95 2005.02  326.67 2008.97
#Mann= 4 ,-1 , 0
       0     .08       0  157.05     .05       0  167.76     .05       0
  219.05     .08       0
Bank Sta=157.05,167.76
Exp/Cntr=0.3,0.1

Type RM Length L Ch R = 1 ,1879    ,149.79,149.59,149.21
XS GIS Cut Line= 2
  951623.2676945  763261.6359924  951385.9710542  763127.7418482
#Sta/Elev= 30
       0 2016.48   19.95 2004.06   28.33 1997.22   37.17 1993.31    47.4 1985.98
   67.21 1976.63   72.92 1972.82   80.56 1972.25    84.3 1972.53   88.49 1971.71
   95.15 1966.18    98.4 1966.45  103.81 1966.14  109.54 1965.54  116.17 1965.53
  125.01 1965.57  130.66 1965.65  136.59 1967.88  142.26 1968.69  158.27 1972.04
  166.89 1973.57  178.94 1976.71  194.48 1978.69  198.71 1979.59  223.09 1987.05
  229.85 1988.61  244.54 1993.18  252.25 1995.29  259.08 1996.66  272.46 2000.02
#Mann= 4 ,-1 , 0
       0     .05       0  103.81     .05       0  125.01     .07       0
  166.89     .05       0
Bank Sta=103.81,125.01
Exp/Cntr=0.3,0.1

Type RM Length L Ch R = 1 ,1731    ,104.54,108.3,114.65
XS GIS Cut Line= 4
  951811.2362068  763211.9791603  951640.8723025  763102.8013042
  951557.1889744  763051.5449841  951395.0529102  763029.5781361
#Sta/Elev= 30
       0 2011.63   12.64 2003.81   19.39  1998.6   27.54 1996.88   30.36 1993.92
   38.75 1991.01   76.13 1990.88  145.27 1991.13  177.13 1989.66  193.49 1982.27
  205.78 1972.88   207.4 1971.26  214.25 1970.55  220.38 1968.79  238.53 1965.17
  243.76 1964.02  251.49 1963.61  259.03 1964.26  262.28 1965.36  273.56 1969.83
  285.53 1972.28  301.57 1975.16  330.73 1978.68  359.59  1981.3   365.8  1982.4
  397.79 1985.72  425.32 1992.93  430.14 1993.17  446.52 1998.98  464.09 2003.44
#Mann= 6 ,-1 , 0
       0     .09       0   30.36     .03       0   76.13     .07       0
  238.53     .05       0  262.28     .07       0  330.73     .05       0
Bank Sta=238.53,262.28
Exp/Cntr=0.3,0.1

Type RM Length L Ch R = 1 ,1622    ,384.75,373.95,363.8
XS GIS Cut Line= 4
  951828.6155348  763044.8726001  951676.2146386   762976.693656
  951589.3190225   762984.714648  951402.1594702  762911.1873519
#Sta/Elev= 30
       0 2020.91   19.03 2000.45      27 1994.55   36.79 1990.33   53.93 1989.31
   98.11  1988.4  118.65 1987.61   133.3 1986.59  141.56 1985.44  147.14 1985.41
  148.19 1985.31  163.03 1977.78  166.96 1974.78  172.11  1969.7  177.57 1966.35
  184.85  1964.8  191.08 1962.62  205.93 1963.45  209.73 1963.93  212.14  1964.9
  217.28 1965.98  235.27 1972.35  255.39 1973.57  261.44 1974.48  285.11 1976.85
  372.09 1982.69   393.6 1984.83  435.89 1989.96  451.73 1993.68  455.31 1995.14
#Mann= 5 ,-1 , 0
       0      .1       0   98.11     .03       0  147.14     .06       0
  184.85     .05       0  212.14     .05       0
Bank Sta=184.85,212.14
Exp/Cntr=0.3,0.1
