HEC-RAS study lds_big_laurel_crk.prj: lds_big_laurel_crk

--- lds_big_laurel_crk.g20 (geometry) --- (continued)

Type RM Length L Ch R = 1 ,116099  ,303.61,273.89,253.97
BEGIN DESCRIPTION:
116020.6
END DESCRIPTION:
XS GIS Cut Line= 6
  931887.6662857  804929.7234019  931832.9783805  805033.0217541
  931819.3066603  805102.9002319  931816.2689554  805125.6860909
  931817.7878079  805172.7787097   931814.750103  805230.5043197
#Sta/Elev= 29
       0 2463.34    7.81    2463      21 2456.04   38.08 2446.91   40.87  2445.5
   51.04 2441.82   53.73 2440.92   64.58 2439.24   68.86 2439.19   82.91 2439.35
   97.04 2439.63  124.21 2439.85  136.36 2440.17  148.49 2440.13   160.1 2439.74
  162.63 2439.74  171.09 2439.17  175.852438.187     180 2437.33  193.69 2435.72
  210.57 2437.95  231.58 2439.51  240.65  2439.6  248.36 2440.24  266.53 2444.41
  271.47 2446.07  272.28 2446.59  283.11 2456.51     316 2481.28
#Mann= 3 , 0 , 0
       0    .075       0  175.85     .05       0  210.57    .075       0
#Block Obstruct= 1 ,-1
    10.5    41.62487.924
Bank Sta=175.85,210.57
Exp/Cntr=0.5,0.3

Type RM Length L Ch R = 1 ,115825  ,98.38,105.67,97.52
XS GIS Cut Line= 4
  931530.1726676  804851.8327983  931592.1547514  805198.3728582
  931596.6631725  805252.4667415  931630.4712094  805409.1133771
#Sta/Elev= 30
       0 2457.94   77.94 2450.48   81.33 2450.71   86.55 2448.84  103.77 2440.88
  125.29 2438.54  149.87 2438.02  169.08 2432.43  188.75 2427.67  203.79 2427.12
  213.79 2428.98  233.35  2434.5  268.92 2435.75  305.64 2439.39  324.58    2439
  337.15 2437.46  349.71 2433.81  355.12 2432.82  361.26  2431.7  381.34 2430.76
  401.61 2430.86  410.08 2432.84  436.69 2440.35  451.57 2442.04  471.06 2447.05
  504.33 2465.64  513.54 2466.34  527.51 2470.76  541.68 2474.25  566.57 2483.65
#Mann= 3 , 0 , 0
       0     .06       0  355.12     .05       0  410.08    .075       0
#XS Ineff= 2 , 0
       0     335    2438     427       0    2438
Permanent Ineff=
       F       F
Bank Sta=355.12,410.08
Exp/Cntr=0.5,0.3

Type RM Length L Ch R = 3 ,115764  ,,,
Bridge Culvert--1,0,-1,-1, 0
Deck Dist Width WeirC Skew NumUp NumDn MinLoCord MaxHiCord MaxSubmerge Is_Ogee
44,12,2.6,0, 6, 6, , , 0.95, 0, 1,1,,
       0     345     345     417     417     555
    2438    2438    2438    2438    2438    2438
                    2436    2436
       0     410     410     482     482     620
    2438    2438    2438    2438    2438    2438
                    2436    2436
BR Coef=-1 , 0 , 0 ,, 0 ,,,0.8,-1,,0,
WSPro=,,,, 1 ,,,, 0 ,,,, 0 ,,,,-1 ,-1 ,-1 , 0 , 0 , 0 , 0 , 0
BC Design=,, 0 ,, 0 ,,,,,,

Type RM Length L Ch R = 1 ,115719  ,191,151.6,94.33
XS GIS Cut Line= 3
  931423.1114942  804857.4678125  931532.1974628  805318.6120992
  931562.8541114  805460.3907774
#Sta/Elev= 30
       0 2452.03   30.13 2452.51   50.19 2451.95   74.57 2449.47   83.09  2445.6
  103.04 2437.86   116.2  2435.3  120.17 2433.81  133.93  2430.6  146.09    2429
  168.51 2427.47  238.39 2426.44   278.6 2426.94  333.46 2429.16  362.83 2432.25
  396.94 2434.94  409.38 2436.96  417.89 2436.39  421.84 2431.38  433.77 2429.21
  442.04 2429.22  464.03 2430.13  476.11 2432.56  481.74 2433.71  498.33 2442.89
  508.89 2443.23  547.84 2447.23  569.28 2458.77  577.88 2461.91  618.93 2486.08
#Mann= 3 , 0 , 0
       0     .06       0  421.84     .05       0  476.11     .08       0
#XS Ineff= 2 , 0
       0     395    2433     497       0    2433
Permanent Ineff=
       F       F
Bank Sta=421.84,476.11
Exp/Cntr=0.5,0.3

Type RM Length L Ch R = 1 ,115567  ,651.69,486.48,462.07
BEGIN DESCRIPTION:
115489.5
END DESCRIPTION:
XS GIS Cut Line= 6
  931242.5329471  804933.5282143  931229.3302993   805000.420196
  931377.2499345   805321.649804  931412.1886613  805412.7963126
  931436.4943969  805441.6586055  931517.0068901  805491.7889291
#Sta/Elev= 30
       0 2436.47    3.03    2436   27.61    2427    42.3 2425.76   73.73  2425.1
  109.77  2425.3  185.96 2424.74  213.26 2423.86  234.38 2422.42  252.88 2424.25
  283.16 2425.21  306.46 2425.17  343.31 2424.21  395.83 2425.21  434.19 2427.46
  461.56 2431.24  466.15 2430.62  478.63 2426.17  481.95  2425.7  498.25 2424.31
  506.14 2425.66  533.51 2429.96  554.37 2430.21  565.96 2431.57  580.51 2440.63
  593.54 2446.16  603.35 2446.48  610.72 2446.15  621.12 2446.83  652.08 2475.56
#Mann= 3 , 0 , 0
       0     .06       0  481.95     .05       0  506.14    .075       0
Bank Sta=481.95,506.14
Exp/Cntr=0.3,0.1

Type RM Length L Ch R = 1 ,115081  ,442.88,472.96,479.55
BEGIN DESCRIPTION:
115003.0
END DESCRIPTION:
XS GIS Cut Line= 6
  930638.9688483  805617.8741645  930777.2059273  805630.0270323
  930892.6571472  805646.7364574  931094.6972943   805728.767803
  931138.7511841  805768.2651355  931217.7448248  805803.2038623
#Sta/Elev= 30
       0 2435.22    3.05  2433.3   23.37 2427.15   36.31  2422.6   52.79 2420.28
   86.49  2420.2  108.96 2418.39  125.73 2420.75  132.66 2421.12  242.18 2423.19
  274.32 2422.68  305.37 2422.86   361.4 2421.85  403.58    2422  423.67 2419.42
   441.5 2417.15  454.21 2419.31  468.36 2422.23  481.65  2423.8  487.25 2425.79
  509.17 2427.56  523.38 2427.23  541.06 2428.97  543.67 2430.32  556.38    2439
  560.13 2440.92  566.97 2442.88   585.7 2449.97  606.18 2458.92  619.03 2462.12
#Mann= 3 , 0 , 0
       0     .06       0  423.67     .05       0  454.21    .075       0
Bank Sta=423.67,454.21
Exp/Cntr=0.3,0.1

Type RM Length L Ch R = 1 ,114608  ,120.54,132.6,166.33
BEGIN DESCRIPTION:
114530.0
END DESCRIPTION:
XS GIS Cut Line= 6
    930561.49406  806024.9921635  930590.3573771  806038.6638837
  930699.7321631    806046.25917  930801.5116629    806103.98478
  930836.4514139   806113.099943  930948.8639048  806192.0925595
#Sta/Elev= 30
       0 2447.46      14 2443.29    38.9 2438.28   44.43  2435.1   53.75 2430.62
   57.39 2427.99   59.64 2427.33   70.06 2421.94    82.1 2418.66   95.68 2413.21
  105.55 2412.55  130.53    2414  147.38 2413.89  198.18 2414.97  214.06 2413.89
  217.292413.376  226.31 2411.94  243.64  2410.7  249.91 2410.69   266.2 2413.22
  281.27 2414.86  328.33 2417.07  369.01 2416.92  371.36 2417.31  383.99 2421.02
     394 2424.69  415.83 2435.53  425.04 2442.71  430.98  2446.5  432.61 2447.77
#Mann= 3 , 0 , 0
       0     .06       0  217.29     .05       0   266.2     .08       0
#Block Obstruct= 2 ,-1
  197.82  210.442425.734  112.01  144.142423.868
Bank Sta=217.29,266.2
Exp/Cntr=0.5,0.3

Type RM Length L Ch R = 1 ,114475  ,29.76,38.06,22.2
BEGIN DESCRIPTION:
114397.4
END DESCRIPTION:
XS GIS Cut Line= 5
  930588.8385246   806078.160192  930620.7395466  806137.4056786
  930686.0604429  806182.9784208  930751.3813392  806231.5888678
  930822.7786695  806309.0636561
#Sta/Elev= 30
       0 2436.41    7.53 2434.84   14.78 2432.72   20.62 2430.45   23.34 2429.58
   32.99 2424.31   36.11  2422.2   37.41 2421.64    55.7 2416.87   57.21 2416.09
   74.69 2414.72   79.98 2414.47   83.07 2413.88   95.58 2413.55  100.89 2413.22
  125.07 2412.87  151.56 2412.85  164.49 2412.98  185.61 2410.93  201.84 2409.24
  215.01 2412.32  227.84  2413.9  248.59 2413.39  260.44 2413.41  268.93  2413.7
  283.85 2418.65  305.61 2427.29  326.74 2436.61  331.62 2438.01  333.72 2439.01
#Mann= 3 , 0 , 0
       0     .07       0  185.61     .05       0  215.01     .07       0
#XS Ineff= 2 , 0
       0  176.16 2416.99  221.16       0 2416.99
Permanent Ineff=
       F       F
#Block Obstruct= 2 ,-1
   50.83  108.642433.241  145.96  162.032422.981
Bank Sta=185.61,215.01
Exp/Cntr=0.5,0.3

Type RM Length L Ch R = 3 ,114457  ,,,
Node Photo=H:\PROJ\06-0741\CE\GIS\DATA\FRENCH_BROAD_RIVER\SHAPEFILES\survey_data\photos\FBSTR_1251.JPG
BEGIN DESCRIPTION:
114381.5  FBSTR_1251
END DESCRIPTION:
Bridge Culvert--1,0,-1,-1, 0
Deck Dist Width WeirC Skew NumUp NumDn MinLoCord MaxHiCord MaxSubmerge Is_Ogee
9,14,2.6,0, 7, 7, , , 0.95, 0, 1,1,,
   36.33  186.16  186.16  198.66  211.16  211.16  277.86
 2416.79 2416.99 2416.99 2416.99 2416.99 2416.99 2416.66
                 2415.99 2415.99 2415.99
   36.07  188.75  188.75  201.25  213.75  213.75  271.17
 2416.93 2416.99 2416.99 2416.99 2416.99 2416.99 2416.75
                 2415.99 2415.99 2415.99
BR Coef=-1 , 0 , 0 ,, 0 ,,,0.8,0,,0,
WSPro=,,,, 1 ,,,, 0 ,,,, 0 ,,,,-1 ,-1 ,-1 , 0 , 0 , 0 , 0 , 0
BC Design=,, 0 ,, 0 ,,,,,,

Type RM Length L Ch R = 1 ,114437  ,162.02,228.82,276.88
BEGIN DESCRIPTION:
114359.4
END DESCRIPTION:
XS GIS Cut Line= 6
  930570.6092229  806102.4659276  930585.7997956  806145.0009649
  930692.1368768  806234.6275968  930745.3049053  806274.1239051
  930787.8399426  806302.9872222  930804.5503919  806324.2542288
#Sta/Elev= 30
       0 2433.74    5.25 2431.78    16.2 2425.93   24.78 2421.72   33.58 2418.26
   38.82 2415.46   45.17 2415.01   73.55 2414.35   86.93 2413.44    93.4  2413.4
  111.09 2412.68  144.81 2412.62  150.03 2412.44  157.12 2411.28   162.8 2410.82
  166.09 2411.31  170.44  2410.7  175.852410.296  182.78 2409.84  198.36 2409.28
  201.25 2408.74  212.26 2409.02  219.05  2410.3   220.6 2410.41  235.83 2413.66
  258.64 2412.48  286.69 2422.03  301.88 2426.83  308.67 2428.67  328.92 2438.32
#Mann= 3 , 0 , 0
       0    .065       0  175.85     .05       0  219.05     .07       0
#XS Ineff= 2 , 0
       0  173.35    2413  228.75       0    2413
Permanent Ineff=
       F       F
#Block Obstruct= 2 ,-1
   40.83  101.822427.439  150.14  167.282423.695
Bank Sta=175.85,219.05
Exp/Cntr=0.5,0.3

Type RM Length L Ch R = 1 ,114208  ,258.49,246.22,152.68
BEGIN DESCRIPTION:
114130.5
END DESCRIPTION:
XS GIS Cut Line= 5
  930415.6606705  806099.4282227  930441.4852585  806199.6878459
  930479.4627144  806275.6427576  930526.5553332  806391.0950017
  930570.6092229  806480.7216336
#Sta/Elev= 30
       0 2440.51    1.01 2439.87    3.54  2437.7   23.72 2418.83   27.46 2417.79
   37.99 2414.11   49.62 2412.89   70.03  2412.3  111.73 2411.63     136 2411.68
  152.09 2411.09  168.85 2410.84  190.47 2410.82  202.65 2410.54  245.02 2409.18
  265.71 2408.75  284.57 2407.16  290.71 2406.45  308.86 2405.53  315.79 2405.55
  319.062407.291  327.82 2412.31  329.83 2411.98  334.44 2411.93  337.89 2412.48
  342.21 2414.18  350.92 2416.84  382.27 2431.82  408.87 2437.49  413.01 2438.14
#Mann= 3 , 0 , 0
       0     .06       0  284.57     .05       0  319.06    .075       0
#Block Obstruct= 1 ,-1
  392.43  413.012448.141
Bank Sta=284.57,319.06
Exp/Cntr=0.3,0.1

Type RM Length L Ch R = 1 ,113962  ,112.46,129.57,144.03
BEGIN DESCRIPTION:
113884.3
END DESCRIPTION:
XS GIS Cut Line= 5
  930175.6440918   806254.375751  930254.6367083  806397.1704114
  930289.5764593  806460.9734795  930364.0114944  806509.5839265
  930488.5778773  806555.1566687
#Sta/Elev= 30
       0 2420.18   61.47 2416.49   80.05 2414.65  105.62 2412.93  211.74 2407.63
  223.24 2405.18  227.08 2403.93  228.97 2403.62  233.49 2402.89   238.1 2401.75
  245.89  2401.4  253.55 2403.41  258.482404.185  270.53 2406.27  287.68 2406.59
  299.21 2406.37  307.71 2408.38  312.33 2408.88  335.15 2408.67  339.76 2409.34
  361.31 2410.68  368.74 2411.87  376.89 2412.82  381.06 2413.82  391.84 2419.83
  402.81 2423.75  410.12 2425.04  425.69 2428.92  434.65 2430.37  457.47  2434.8
#Mann= 3 , 0 , 0
       0     .05       0  228.97     .05       0  258.48     .07       0
#Block Obstruct= 2 ,-1
   96.69   169.52427.218  442.33  457.472444.801
Bank Sta=228.97,258.48
Exp/Cntr=0.5,0.3

Type RM Length L Ch R = 1 ,113833  ,140.15,43.43,50.25
BEGIN DESCRIPTION:
113754.7
END DESCRIPTION:
XS GIS Cut Line= 6
  930106.6771303  806329.0524915  930159.4109083  806461.9945826
  930203.1606179  806558.8693053  930237.5360481  806596.3694953
  930318.7859478  806643.2449889  930450.0361007  806694.8071101
#Sta/Elev= 30
       0 2418.95    6.31 2417.97   14.07 2414.36   32.74 2415.62   39.16  2414.6
      70 2412.35   77.82 2412.16  111.51 2409.81  144.07 2407.98  207.63 2406.02
  216.162403.499  224.86 2401.09  241.38 2400.84  253.91 2403.18  261.77 2404.43
  287.75 2405.94  333.77 2406.07  362.61 2406.59  370.33  2407.1  380.35 2406.66
  392.89 2407.07  412.08    2409  418.83 2409.16  431.04 2411.57  443.71 2414.88
  455.32 2417.18  472.01 2422.89  504.18 2429.03  520.77 2433.19     535 2437.18
#Mann= 3 , 0 , 0
       0    .055       0  216.16     .05       0  253.91    .055       0
#XS Ineff= 2 , 0
       0  213.16 2407.93  258.16       0 2407.93
Permanent Ineff=
       F       F
#Block Obstruct= 2 ,-1
  373.64  425.132420.477   95.15  141.522424.049
Bank Sta=216.16,253.91
Exp/Cntr=0.5,0.3

Type RM Length L Ch R = 3 ,113814  ,,,
Node Photo=H:\PROJ\06-0741\CE\GIS\DATA\FRENCH_BROAD_RIVER\SHAPEFILES\survey_data\photos\FBSTR_1254.JPG
BEGIN DESCRIPTION:
113738.5  FBSTR_1254
END DESCRIPTION:
Bridge Culvert--1,0,-1,-1, 0
Deck Dist Width WeirC Skew NumUp NumDn MinLoCord MaxHiCord MaxSubmerge Is_Ogee
9,9,2.6,0, 7, 7, , , 0.95, 0, 1,1,,
       0  223.16  223.16  245.16  248.16  248.16  420.76
 2407.92 2407.93 2407.93 2407.93 2407.93 2407.93 2407.86
                 2406.93 2406.93 2406.93
   12.03   124.5   124.5     137   149.5   149.5  320.19
 2407.88 2407.93 2407.93 2407.93 2407.93 2407.93  2407.7
                 2406.93 2406.93 2406.93
BR Coef=-1 , 0 , 0 ,, 0 ,,,0.8,0,,0,
WSPro=,,,, 1 ,,,, 0 ,,,, 0 ,,,,-1 ,-1 ,-1 , 0 , 0 , 0 , 0 , 0
BC Design=,, 0 ,, 0 ,,,,,,

Type RM Length L Ch R = 1 ,113789  ,181.6,162.32,83.29
BEGIN DESCRIPTION:
113711.3
END DESCRIPTION:
XS GIS Cut Line= 6
  930037.5360589   806547.932134  930121.9107183  806552.6197857
  930153.1613887  806566.6827411  930187.5357948  806599.4942551
  930268.7856944  806661.9945718  930420.3483223   806751.056883
#Sta/Elev= 30
       0 2443.08   11.59 2432.01   34.01 2411.95   40.92 2407.28   48.09 2405.83
   71.78 2405.05   98.02 2405.03  115.58 2402.83   118.8 2402.69  120.74  2402.5
  126.75 2400.82  139.14 2400.85  157.31 2402.57   167.1 2403.81  198.49 2405.45
  223.38 2404.66  248.23  2404.9  257.84 2405.17  299.69 2405.11  324.09 2405.76
  346.37 2407.32  359.69 2410.18  369.15 2413.04  375.06 2415.21  395.65 2427.82
  402.61 2429.74  412.48 2432.97  422.42 2436.88  432.79 2439.87  444.62 2442.58
#Mann= 3 , 0 , 0
       0    .065       0   118.8     .05       0  157.31    .055       0
#XS Ineff= 2 , 0
       0   109.5    2404   164.5       0    2404
Permanent Ineff=
       F       F
#Block Obstruct= 1 ,-1
  294.48  340.162416.797
Bank Sta=118.8,157.31
Exp/Cntr=0.5,0.3

Type RM Length L Ch R = 1 ,113627  ,175.43,150.42,48.34
BEGIN DESCRIPTION:
113549.0
END DESCRIPTION:
XS GIS Cut Line= 5
  930040.6608187  806729.1825403  930093.7858318  806730.7444081
  930173.4738636  806733.8701921  930275.0362382  806766.6827303
  930364.0985493  806807.3076801
#Sta/Elev= 30
       0 2433.43    2.34 2431.43    19.6 2417.94   23.69 2415.16   38.03 2407.16
    47.52402.094   54.84 2398.17   63.31 2398.49   73.31 2400.41   84.68 2401.95
   93.62 2402.08   95.83 2402.33  101.19 2402.46  106.01 2402.38  115.32 2402.61
  143.69 2402.08  175.84  2402.7   188.9 2402.58  211.84  2402.9  216.03 2402.83
  223.67 2403.03  228.95 2402.92   264.4 2404.25  272.06    2405  284.23 2406.82
  285.59 2407.71  296.33 2413.65  303.36 2417.93  324.64 2430.41  337.52 2433.25
#Mann= 3 , 0 , 0
       0     .07       0    47.5     .05       0   84.68     .06       0
Bank Sta=47.5,84.68
Exp/Cntr=0.5,0.3

Type RM Length L Ch R = 1 ,113476  ,50.81,57.77,61.12
BEGIN DESCRIPTION:
113398.6
END DESCRIPTION:
XS GIS Cut Line= 6
  930020.3483438  806888.5575797  930067.2238374  806907.3071626
  930095.3487238  806904.1824028  930204.7235099  806838.5573264
  930265.6609346  806832.3067826  930373.4738529  806852.6192575
#Sta/Elev= 30
       0 2436.37   18.23 2426.79   23.94 2423.24   31.54 2419.02   42.64 2412.31
   50.49 2408.48   73.59 2399.08   97.95 2397.77  117.73 2395.99  135.42 2398.66
  140.25  2399.4  153.47 2400.22  162.78 2400.15  207.74 2401.63  215.02 2401.53
  221.56 2401.71  231.12 2401.69  254.13 2402.06  268.71 2402.73  274.81 2403.14
  289.68 2404.61  299.04 2406.72  307.96 2409.95  315.62 2413.77  319.98  2415.3
  326.53 2417.87  333.29 2421.46  347.05 2426.61  354.78  2429.3  380.29 2435.38
#Mann= 3 , 0 , 0
       0     .08       0   97.95     .05       0  135.42     .06       0
#XS Ineff= 2 , 0
       0    94.8 2401.94   140.8       0 2401.94
Permanent Ineff=
       F       F
Bank Sta=97.95,135.42
Exp/Cntr=0.5,0.3

Type RM Length L Ch R = 3 ,113450  ,,,
Node Photo=H:\PROJ\06-0741\CE\GIS\DATA\FRENCH_BROAD_RIVER\SHAPEFILES\survey_data\photos\FBSTR_1260A.JPG
BEGIN DESCRIPTION:
113365.6  FBSTR_1260A
END DESCRIPTION:
Bridge Culvert--1,0,-1,-1, 0
Deck Dist Width WeirC Skew NumUp NumDn MinLoCord MaxHiCord MaxSubmerge Is_Ogee
16,18,2.6,0, 7, 7, , , 0.95, 0, 1,1,,
       0   104.8   104.8   117.8   130.8   130.8  253.01
 2401.94 2401.94 2401.94 2401.94 2401.94 2401.94 2401.95
                 2400.44 2400.44 2400.44
       0   109.2   109.2   122.2   135.2   135.2  282.03
 2401.94 2401.94 2401.94 2401.94 2401.94 2401.94 2401.85
                 2400.44 2400.44 2400.44
BR Coef=-1 , 0 , 0 ,, 0 ,,,0.8,0,,0,
WSPro=,,,, 1 ,,,, 0 ,,,, 0 ,,,,-1 ,-1 ,-1 , 0 , 0 , 0 , 0 , 0
BC Design=,, 0 ,, 0 ,,,,,,

Type RM Length L Ch R = 1 ,113419  ,178.09,170.38,210.2
BEGIN DESCRIPTION:
113340.8
END DESCRIPTION:
XS GIS Cut Line= 6
  930004.7235207  806929.1825295  930101.5982434   806957.307416
  930157.8490405  806921.3701179  930201.5987501  806907.3071626
  930318.7859478  806885.4317957  930364.0985493  806897.9318591
#Sta/Elev= 30
       0 2434.99     9.7 2430.08   29.92 2417.82   37.17 2412.15   40.93 2409.63
   55.02 2403.51   57.02 2402.36   66.08 2401.26   83.48 2400.11  101.75 2398.11
  109.28  2396.7  130.86 2396.42  146.83 2397.49  150.26 2397.28  159.09 2398.29
  169.58 2399.16  188.66 2399.13  251.71 2400.75  280.35 2401.77   287.4 2402.37
  298.28 2403.63  300.38 2404.33  313.19 2413.65  317.84 2416.73  323.26 2419.51
  332.76 2422.84  340.21 2424.48   356.2 2429.01  367.09 2431.78  380.68 2435.64
#Mann= 3 , 0 , 0
       0     .08       0  101.75     .05       0  146.83     .07       0
#XS Ineff= 2 , 0
       0    94.2    2399   150.2       0    2399
Permanent Ineff=
       F       F
Bank Sta=101.75,146.83
Exp/Cntr=0.5,0.3

Type RM Length L Ch R = 1 ,113248  ,145.02,192.32,217.82
BEGIN DESCRIPTION:
113170.4
END DESCRIPTION:
XS GIS Cut Line= 6
  929967.2233307  807104.1823921  930075.0362489  807133.8701705
  930121.9107183  807113.5576956  930204.7235099  807097.9318483
  930292.2239533  807101.0576323  930325.0364915  807108.8700438
#Sta/Elev= 30
       0 2438.89    7.57 2439.57    9.84 2438.28    13.1 2435.41   21.19 2431.98
   44.41 2424.21   61.46 2421.04   71.67 2418.25   77.51 2415.11   90.01 2411.74
   97.84 2411.01  103.97  2409.3  111.91 2407.89  146.44 2402.74  167.87 2394.63
  178.31 2393.23  182.07 2392.37  190.91 2393.69  199.05 2394.06  213.68 2395.98
  220.71 2396.56   250.9 2397.69  255.77 2397.47  275.93 2399.78  282.73 2399.99
  309.72 2419.61  317.48 2424.43  326.76 2429.38  340.15 2435.18  368.69 2445.77
#Mann= 3 , 0 , 0
       0    .075       0  167.87     .05       0  199.05     .07       0
#Block Obstruct= 1 ,-1
   91.13  141.082429.687
Bank Sta=167.87,199.05
Exp/Cntr=0.5,0.3

Type RM Length L Ch R = 1 ,113056  ,25.95,41.23,40.86
BEGIN DESCRIPTION:
112978.1
END DESCRIPTION:
XS GIS Cut Line= 6
  930000.0358689  807249.4944762  930062.5361856  807277.6193626
  930107.8487872  807286.9946662  930209.4111617  807305.7442491
  930225.0359848  807310.4319009  930281.2857577  807332.3072678
#Sta/Elev= 30
       0 2417.44    3.95 2415.98    12.8 2415.45   25.06 2413.44   34.38 2411.54
   51.86 2406.38   56.03 2405.61   77.02 2400.55   90.47 2398.76  109.34 2397.42
  143.82 2396.77  159.452393.435  164.24 2392.35  171.16 2390.21  183.87 2392.41
   187.2 2393.22  197.49 2395.54  198.03    2396  205.06 2398.08  211.62 2398.29
  215.75  2399.1  223.83 2398.93  232.29  2404.9  237.71 2410.12  239.44 2412.03
  250.08 2422.19   256.4  2426.9  257.89  2427.9  283.16 2441.88  294.75 2447.81
#Mann= 3 , 0 , 0
       0     .07       0  159.45     .05       0   187.2    .075       0
#XS Ineff= 2 , 0
       0  146.95 2398.53  200.95       0 2398.53
Permanent Ineff=
       F       F
#Block Obstruct= 1 ,-1
   59.31   91.242420.832
Bank Sta=159.45,187.2
Exp/Cntr=0.5,0.3

Type RM Length L Ch R = 3 ,113035  ,,,
Node Photo=H:\PROJ\06-0741\CE\GIS\DATA\FRENCH_BROAD_RIVER\SHAPEFILES\survey_data\photos\FBSTR_1260.JPG
BEGIN DESCRIPTION:
112956  FBSTR_1260
END DESCRIPTION:
Bridge Culvert--1,0,-1,-1, 0
Deck Dist Width WeirC Skew NumUp NumDn MinLoCord MaxHiCord MaxSubmerge Is_Ogee
14,12,2.6,0, 7, 7, , , 0.95, 0, 1,1,,
   93.61  156.95  156.95  168.95  190.95  190.95  212.15
 2398.52 2398.53 2398.53 2398.53 2398.53 2398.53 2398.39
                 2396.53 2396.53 2396.53
    85.5  159.24  159.24  176.24  193.24  193.24  200.62
 2398.53 2398.53 2398.53 2398.53 2398.53 2398.53 2398.45
                 2396.53 2396.53 2396.53
BR Coef=-1 , 0 , 0 ,, 0 ,,,0.8,0,,0,
WSPro=,,,, 1 ,,,, 0 ,,,, 0 ,,,,-1 ,-1 ,-1 , 0 , 0 , 0 , 0 , 0
BC Design=,, 0 ,, 0 ,,,,,,

Type RM Length L Ch R = 1 ,113015  ,188.06,195.51,221.81
BEGIN DESCRIPTION:
112936.9
END DESCRIPTION:
XS GIS Cut Line= 6
  929995.3482171  807277.6193626   930053.160882  807301.0576215
  930118.7859585  807332.3072678  930181.2862752  807341.6825713
  930207.8482697  807347.9320909  930254.7237633   807365.119806
#Sta/Elev= 30
       0 2416.64    4.49 2415.78   12.34 2415.48   21.79 2412.26   32.14 2409.98
   44.96 2406.26   54.32 2403.07   67.07  2400.4   79.11 2398.92   98.35 2397.34
  124.31 2396.25  145.89 2396.17  151.61 2395.83  158.76 2394.21  164.782391.438
  166.08 2390.84  183.67 2389.24  189.01 2390.19  191.08 2391.86  194.52 2394.71
  200.62 2398.45  209.45 2398.49  215.53 2399.46  221.38 2398.93  224.78 2400.24
     234 2406.62  242.95 2415.44  247.19 2419.17  259.61 2431.06  275.49 2439.03
#Mann= 3 , 0 , 0
       0     .07       0  164.78     .05       0  191.08    .075       0
#XS Ineff= 2 , 0
       0  149.24    2394  203.24       0    2394
Permanent Ineff=
       F       F
#Block Obstruct= 1 ,-1
   51.48   91.522420.153
Bank Sta=164.78,191.08
Exp/Cntr=0.5,0.3

Type RM Length L Ch R = 1 ,112819  ,167.92,165.01,124.48
BEGIN DESCRIPTION:
112741.3
END DESCRIPTION:
XS GIS Cut Line= 6
   929906.285906  807472.9327243  929987.5358056  807472.9327243
  930023.4731036  807485.4317634  930065.6609454  807507.3071303
  930118.7859585  807547.9320801  930159.4109083  807566.6826872
#Sta/Elev= 30
       0 2415.63   13.33 2411.52   19.86 2409.96   28.91 2407.42   41.79  2404.4
   44.88 2403.79   57.54 2401.65   81.71 2398.04   97.41 2395.32   98.46 2394.93
  105.07 2393.73  118.53 2392.48  136.91 2391.19  144.09  2390.2   157.9 2386.76
  170.21 2387.61  171.36 2387.49   176.7 2388.36  181.95 2389.22  188.09 2390.67
  189.07 2391.15  199.31 2394.89  201.23 2394.86   211.6 2396.54   224.6 2402.78
  227.35 2404.52  234.96  2410.3  254.22 2423.26  269.79 2436.13  278.49  2441.6
#Mann= 3 , 0 , 0
       0     .07       0  144.09     .05       0   176.7    .075       0
#Block Obstruct= 1 ,-1
   72.95   95.782413.162
Bank Sta=144.09,176.7
Exp/Cntr=0.3,0.1

Type RM Length L Ch R = 1 ,112654  ,368.15,334.24,284.16
BEGIN DESCRIPTION:
112576.3
END DESCRIPTION:
XS GIS Cut Line= 6
   929851.599025  807627.6201119  929910.9735577  807629.1819797
  929959.4109191  807636.9943913  930007.8482805  807652.6202386
  930046.9113625  807657.3068662  930112.5364389  807647.9325868
#Sta/Elev= 30
       0 2426.14    4.84 2424.59   12.08 2421.88   21.21 2419.56   28.67 2416.86
   48.85 2410.72   52.93 2409.75   59.71 2409.36   88.64 2393.01   100.2  2387.7
  103.722387.167  111.16 2385.93  128.11 2385.54  137.162387.178  151.17 2389.43
  158.98 2389.72     165 2389.57  179.51 2389.84  186.68 2392.71  193.77 2394.81
   195.3 2395.08  200.37 2396.89  210.09 2401.74  214.76 2403.33  218.77 2406.18
  223.29 2407.83  231.23 2411.37  236.99 2415.22  256.63 2424.14  264.99 2428.67
#Mann= 3 , 0 , 0
       0     .07       0  103.72     .05       0  137.16    .075       0
Bank Sta=103.72,137.16
Exp/Cntr=0.3,0.1

Type RM Length L Ch R = 1 ,112320  ,414.79,419.69,427.76
BEGIN DESCRIPTION:
112242.1
END DESCRIPTION:
XS GIS Cut Line= 5
  929881.2857793  808022.9324386  929954.7232673  807990.1199004
  930004.7235207  807963.5568817  930070.3485972  807944.8072988
  930137.5365656  807922.9319319
#Sta/Elev= 30
       0 2431.04   14.21 2422.02    16.7 2420.59   22.28 2418.63   32.76 2415.44
   40.78 2411.48   48.28 2408.76   62.09 2402.42   62.98 2401.92   70.79 2396.23
   86.91 2385.97      88 2385.13   89.36 2384.42    90.6    2384  100.812383.285
  119.44 2381.93  123.96 2382.33  140.77 2384.37  155.88  2386.2  175.21 2386.35
  200.54 2386.93  206.12 2386.85  210.46 2387.34  222.24 2389.96  228.37 2391.46
  234.86 2393.91  238.84 2395.77  258.17 2407.19  265.96 2410.95  275.96 2416.96
#Mann= 3 , 0 , 0
       0    .075       0  100.81     .05       0  140.77    .075       0
Bank Sta=100.81,140.77
Exp/Cntr=0.3,0.1

Type RM Length L Ch R = 1 ,111900  ,375.81,404.69,382.23
BEGIN DESCRIPTION:
111822.4
END DESCRIPTION:
XS GIS Cut Line= 6
  930001.5987609  808418.2447653  930071.9114891  808388.5569869
  930131.2860219  808366.6826441   930148.473737  808354.1825808
  930192.2234466  808327.6195622  930300.0363648  808321.3700426
#Sta/Elev= 30
       0  2435.8   19.27 2424.31   21.46 2422.55   33.12  2412.8   38.69  2408.3
   40.79 2406.45   45.51  2403.5   65.81 2389.08   80.69 2381.12   84.46 2379.23
  109.95    2380  118.29 2379.28     125 2378.81  143.75 2377.33  156.75 2377.52
  164.31 2378.64  170.25 2379.52   175.4 2380.17  183.63  2380.5  190.08  2381.5
  191.73 2381.84  203.24 2383.33  215.17 2383.93  230.35    2384  246.55 2384.33
  250.84 2384.22  259.82 2384.83  304.42 2409.49  310.02 2412.39  320.05 2415.54
#Mann= 3 , 0 , 0
       0     .07       0     125     .05       0  164.31    .075       0
Bank Sta=125,164.31
Exp/Cntr=0.3,0.1

Type RM Length L Ch R = 1 ,111496  ,170.87,183.57,196.06
BEGIN DESCRIPTION:
111417.7
END DESCRIPTION:
XS GIS Cut Line= 6
  929990.6615895  808730.7443004  930026.5988876  808752.6196673
  930070.3485972  808766.6826226  930160.9738003  808765.1197306
  930281.2857577  808726.0576728  930346.9108342  808661.9944641
#Sta/Elev= 30
       0 2417.43    9.81 2409.63   11.26 2408.73   14.26 2406.13   24.94 2395.47
   37.32 2383.82   39.82 2381.81   59.32 2377.19   80.99 2376.47  152.71 2375.19
  182.42 2375.44  196.13 2375.92  211.312373.228  219.73  2371.6  222.36 2371.97
  241.89 2372.75   258.7 2375.57  274.59 2376.93  278.88 2377.61  284.24 2378.93
  289.87 2381.65   299.6 2385.68  304.52 2386.29  314.13 2388.62  335.95 2389.56
  338.36 2390.03  359.49 2396.41  373.64 2398.62  386.99 2406.78     397 2410.07
#Mann= 3 , 0 , 0
       0     .07       0  211.31     .05       0  241.89     .07       0
#Block Obstruct= 1 ,-1
  148.58  181.682385.428
Bank Sta=211.31,241.89
Exp/Cntr=0.5,0.3

Type RM Length L Ch R = 1 ,111312  ,33.99,45.29,61.4
BEGIN DESCRIPTION:
111234.2
END DESCRIPTION:
XS GIS Cut Line= 6
  929954.7232673  808911.9947067   930018.786476  808936.9948334
  930192.2234466  808936.9948334  930248.4732195  808932.3071816
  930325.0364915  808897.9317514  930404.7234991  808880.7450605
#Sta/Elev= 30
       0 2422.32   12.35 2414.83   16.03 2411.66   26.57 2398.36   34.24 2389.94
    40.7 2388.58   46.43 2388.06   52.16 2385.99   75.05 2374.05   87.03 2373.68
   98.86 2372.73  131.69 2371.81  219.12 2373.33  264.99 2373.04  298.65 2373.37
  308.69  2373.1  322.37 2370.42  323.86 2370.41  335.96 2371.02  344.41 2373.39
  368.03 2380.18  374.07 2381.14  378.15 2380.99  392.79 2389.92  402.73 2390.23
  412.75 2391.68  431.29 2400.93  440.85 2404.73  457.37 2408.18   464.1 2410.61
#Mann= 3 , 0 , 0
       0    .065       0  308.69     .05       0  344.41     .07       0
#XS Ineff= 2 , 0
       0     305    2377     355       0 2378.04
Permanent Ineff=
       F       F
#Block Obstruct= 1 ,-1
  176.95  231.272383.358
Bank Sta=308.69,344.41
Exp/Cntr=0.5,0.3

Type RM Length L Ch R = 3 ,111285  ,,,
Node Photo=H:\PROJ\06-0741\CE\GIS\DATA\FRENCH_BROAD_RIVER\SHAPEFILES\survey_data\photos\FBSTR_1273.JPG
BEGIN DESCRIPTION:
111210.2  FBSTR_1273
END DESCRIPTION:
Bridge Culvert--1,0,-1,-1, 0
Deck Dist Width WeirC Skew NumUp NumDn MinLoCord MaxHiCord MaxSubmerge Is_Ogee
17,10,2.6,0, 7, 7, , , 0.95, 0, 1,1,,
       0     315     315  326.49     345     345  360.89
 2373.37 2378.04 2378.04 2378.04 2378.04 2378.04 2378.08
                 2376.54 2376.54 2376.54
       0     335     335  359.79     365     365  383.55
 2373.42 2378.04 2378.04 2378.04 2378.04 2378.04 2378.11
                 2376.54 2376.54 2376.54
BR Coef=-1 , 0 , 0 ,, 0 ,,,0.8,0,,0,
WSPro=,,,, 1 ,,,, 0 ,,,, 0 ,,,,-1 ,-1 ,-1 , 0 , 0 , 0 , 0 , 0
BC Design=,, 0 ,, 0 ,,,,,,

Type RM Length L Ch R = 1 ,111267  ,229.77,288.87,264.08
BEGIN DESCRIPTION:
111188.9
END DESCRIPTION:
XS GIS Cut Line= 6
   929942.223204  808935.4319414  930028.1607554  808965.1197199
  930157.8490405  808983.8693028  930223.4730928  808979.1826752
  930310.9735362  808954.1825485   930389.098676  808949.4948967
#Sta/Elev= 30
       0 2425.78    2.83 2423.95   17.16 2410.19   24.04 2400.57   27.01 2398.38
   32.73 2397.18   36.44 2395.12   39.63  2394.7   52.08 2390.75   64.06 2382.05
   70.01 2378.11   78.37 2373.32   81.06 2373.57   90.49 2372.94  161.08 2371.79
  239.33 2372.97  282.56  2372.7  312.86 2373.11  329.23 2373.72  339.26 2372.35
  354.19 2370.15  364.85 2370.01  370.04 2372.37  390.72  2381.1  395.11 2382.18
  400.44 2385.68  410.21 2390.16  432.05 2391.74  448.46 2400.73  457.68 2406.26
#Mann= 3 , 0 , 0
       0    .065       0  339.26     .05       0  370.04     .07       0
#XS Ineff= 2 , 0
       0     320    2373     380       0    2373
Permanent Ineff=
       F       F
#Block Obstruct= 1 ,-1
  206.84  231.542382.901
Bank Sta=339.26,370.04
Exp/Cntr=0.5,0.3

Type RM Length L Ch R = 1 ,110978  ,393.27,361.45,399.11
BEGIN DESCRIPTION:
110900.0
END DESCRIPTION:
XS GIS Cut Line= 6
  929954.7232673  809135.4319306  930021.9112358  809197.9322473
  930242.2236999  809243.2448489  930287.5363015  809244.8077409
   930390.661568  809207.3075509  930467.2238158  809210.4323107
#Sta/Elev= 30
       0 2404.23     9.8 2403.62   19.22 2398.27   24.51 2396.39   53.02 2389.69
   67.16 2387.42   75.15 2383.94   84.32 2378.56   92.22 2374.82  100.41 2372.36
  111.32 2370.35  135.51 2368.75  179.12 2369.79  236.88  2369.8  280.19 2371.28
  288.04 2369.04   295.4    2367  323.96 2368.08  348.32 2369.68  373.55 2369.89
  384.97 2375.16  398.19 2383.53  429.59 2386.95  467.17 2394.14  471.49 2395.56
  479.66 2399.77  503.43 2402.59  510.88 2407.74  519.21  2411.6  549.84 2418.64
#Mann= 3 , 0 , 0
       0    .055       0  288.04     .05       0  323.96     .06       0
Bank Sta=288.04,323.96
Exp/Cntr=0.3,0.1

Type RM Length L Ch R = 1 ,110616  ,357.29,436.71,553.88
BEGIN DESCRIPTION:
110538.5
END DESCRIPTION:
XS GIS Cut Line= 6
  929895.3487346  809599.4951178  929989.0986975  809577.6197509
  930051.5990142  809577.6197509  930128.1612621  809585.4321625
  930256.2856311  809613.5570489  930435.9731454  809611.9951811
#Sta/Elev= 30
       0 2413.15   24.27 2380.37   31.51 2371.29   34.17 2368.85   63.17    2366
   69.95 2365.75   99.83 2365.84  113.77 2366.26  169.64 2365.93  205.47 2366.25
   214.5 2365.94  220.032364.655  235.38 2361.35  256.52 2364.18  271.27 2365.76
  277.24  2365.9  400.62 2366.28  410.83 2366.46  426.15 2368.03  430.14 2369.51
  435.92 2371.02  446.36 2374.51  465.42 2382.08  481.39 2387.95  498.22 2393.13
  507.86  2395.3  513.28 2397.64  537.72 2405.91   543.2 2408.14  547.55 2408.49
#Mann= 3 , 0 , 0
       0    .055       0  220.03     .05       0  256.52    .055       0
#Block Obstruct= 1 ,-1
  490.12  539.812416.757
Bank Sta=220.03,256.52
Exp/Cntr=0.3,0.1

Type RM Length L Ch R = 1 ,110180  ,410.03,421.48,385.34
BEGIN DESCRIPTION:
110101.8
END DESCRIPTION:
XS GIS Cut Line= 6
   929812.535943  809885.4326584   929851.599025  809924.4947162
  930051.5990142  810061.9943888  930167.2233199  810161.9948955
  930198.4739903   810168.244415  930248.4732195  810161.9948955
#Sta/Elev= 30
       0 2403.35    6.99 2397.03   20.37 2381.21   45.47 2365.39   51.02 2362.08
   60.23  2358.8   74.47 2357.92   90.22 2355.69  105.93 2357.91   121.5 2359.61
  189.95 2360.03  217.25 2359.25  244.27  2359.3  305.09 2361.06  316.33 2360.18
  335.09 2357.76  360.15 2357.35  371.05    2360  377.42 2363.97  389.79 2370.64
  400.75 2373.18  431.42  2376.1  462.49 2377.74  467.43 2377.54  472.63  2380.8
  477.92 2381.32  481.78 2382.72   487.5 2383.18  509.96 2387.34  533.57 2393.23
#Mann= 3 , 0 , 0
       0     .07       0   74.47     .05       0  105.93    .065       0
#Block Obstruct= 1 ,-1
  321.67  441.992386.693
Bank Sta=74.47,105.93
Exp/Cntr=0.3,0.1

Type RM Length L Ch R = 1 ,109758  ,405.41,431.41,502.46
BEGIN DESCRIPTION:
109680.3
END DESCRIPTION:
XS GIS Cut Line= 6
  929717.2230881  810266.6820298  929756.2861701  810305.7451118
  929807.8482912  810346.3700616  929921.9107291  810408.8693541
  929990.6615895  810452.6200878   930054.723774  810518.2451643
#Sta/Elev= 30
       0  2387.2   13.36 2376.21   29.95 2363.75   39.51 2359.76   47.92 2355.66
   56.38 2355.12   59.23 2355.39   67.63 2354.24   75.19 2352.48   92.68 2353.63
   99.46  2349.9  100.59 2349.57  111.78 2348.37  127.16 2352.28  136.18  2353.5
  144.04 2355.54  166.35 2354.89  199.99 2355.72  277.33 2356.31  300.41 2357.56
  333.39 2360.59  345.71 2363.18  349.52 2365.13  361.57 2372.53   377.5 2375.91
   391.5  2377.2  398.41 2376.37  404.85 2379.47  411.15 2384.07   424.3 2394.95
#Mann= 3 , 0 , 0
       0     .07       0   92.68     .05       0  144.04     .06       0
Bank Sta=92.68,144.04
Exp/Cntr=0.3,0.1

Type RM Length L Ch R = 1 ,109327  ,454.41,432.4,417.75
BEGIN DESCRIPTION:
109248.9
END DESCRIPTION:
XS GIS Cut Line= 6
  929415.6607243  810557.3072222  929470.3486295  810593.2445202
  929510.9735793  810616.6817549  929545.3490095  810685.4326153
  929568.7862442  810736.9947365  929671.9115107   810840.120003
#Sta/Elev= 30
       0 2379.37    6.58 2375.71   21.42 2368.26   23.71 2366.74   27.55 2365.11
   42.04 2357.14   48.58 2354.62   68.78 2351.08  120.95 2352.19  129.892350.299
  149.19 2346.23  163.17 2344.85  182.33 2343.55  186.62 2343.89  193.31 2348.47
  195.17 2350.11  203.27 2349.69  273.23 2348.75  286.92 2348.79   292.7 2349.81
  305.53  2357.3  327.64 2368.37  340.22 2379.28  345.74 2382.63  349.55 2386.04
  353.56 2390.51  358.93 2392.27  366.72 2393.82  385.16 2393.93  391.69 2398.48
#Mann= 3 , 0 , 0
       0     .07       0  129.89     .05       0  195.17     .07       0
Bank Sta=129.89,195.17
Exp/Cntr=0.3,0.1

Type RM Length L Ch R = 1 ,108894  ,224.99,259.67,240.56
BEGIN DESCRIPTION:
108816.5
END DESCRIPTION:
XS GIS Cut Line= 5
  929154.7233104  810915.1193588   929239.098994   810968.244372
  929278.1610518  810997.9321504   929312.536482  811068.2448787
  929332.8489569  811115.1193481
#Sta/Elev= 30
       0 2379.09   20.33  2363.8   33.93 2356.89   41.05 2352.94   49.96  2347.6
   62.73  2345.1   73.61 2343.42   76.78 2341.57   85.05 2337.99    86.2 2337.65
  110.67 2339.13  112.44 2339.54  121.162343.057  123.77 2344.11   127.3 2344.01
  133.13 2344.29  142.15 2344.15  166.17 2342.77  173.73 2342.52  178.99 2342.73
  181.58  2343.3  187.13 2344.91  198.43 2352.46  204.55 2358.08  212.92 2364.46
  222.78 2371.51  231.81 2373.53  239.21 2375.44  255.38 2375.34  278.12 2396.02
#Mann= 3 , 0 , 0
       0     .07       0   76.78     .05       0  121.16     .07       0
Bank Sta=76.78,121.16
Exp/Cntr=0.3,0.1

Type RM Length L Ch R = 1 ,108635  ,83.09,130.31,188.25
BEGIN DESCRIPTION:
108556.9
END DESCRIPTION:
XS GIS Cut Line= 6
  929025.0360494  811022.9322771  929026.5989414   811080.744942
  929039.0990047   811118.245132  929064.0981072  811157.3071898
   929106.285949  811199.4950316  929178.1615693  811240.1199814
#Sta/Elev= 30
       0 2378.03   31.86 2356.61   36.48 2354.47   41.66 2352.91   47.61 2350.55
   61.33 2345.68   81.61 2340.33   86.39 2338.85   89.13 2338.73  110.32 2336.72
  116.94 2336.45  122.29 2335.69  137.08 2335.45  143.63 2335.82   156.1  2335.7
  165.26 2337.12  180.19 2339.27  192.99 2341.43  209.27 2343.04  218.69 2344.85
   231.4 2350.06     242 2358.62  246.94 2361.93  254.41 2367.31  257.26 2368.17
  263.91 2369.57  271.34 2369.62  277.84 2370.36  283.79 2371.88  286.33  2373.6
#Mann= 3 , 0 , 0
       0    .075       0  116.94     .05       0  165.26     .07       0
Bank Sta=116.94,165.26
Exp/Cntr=0.3,0.1

Type RM Length L Ch R = 1 ,108504  ,64.36,80.24,119.24
BEGIN DESCRIPTION:
108426.6
END DESCRIPTION:
XS GIS Cut Line= 6
  928965.6615167  811024.4951691  928937.5356061  811132.3070632
  928937.5356061  811227.6199181  928953.1614534  811276.0572795
  929004.7235745   811376.056762  929028.1608092  811407.3074324
#Sta/Elev= 30
       0 2369.33    2.48 2367.66    7.91 2367.51   43.85 2351.15   48.36 2350.62
   70.11 2342.47   72.37 2342.01   83.38 2341.47  103.78  2338.6   117.9 2337.78
  142.972334.275  151.37 2333.02  164.12 2332.57  177.59 2333.89  206.88 2336.32
  216.25 2336.31  252.08 2337.55  270.38 2338.57  279.11 2342.42  295.49 2347.17
  307.49 2349.22  339.35 2352.88  344.61 2354.18  352.98 2357.83  356.83 2358.99
  367.47 2365.31   386.5 2366.81  398.89 2367.26  401.83  2368.1  409.48 2371.54
#Mann= 3 , 0 , 0
       0    .075       0  142.97     .05       0  177.59     .06       0
#Block Obstruct= 2 ,-1
  244.31  269.362348.461    78.3  104.712354.915
Bank Sta=142.97,177.59
Exp/Cntr=0.5,0.3

Type RM Length L Ch R = 1 ,108424  ,39.46,44.7,38.46
BEGIN DESCRIPTION:
108346.3
END DESCRIPTION:
XS GIS Cut Line= 6
  928918.7860231  811016.6827575  928892.2240286  811058.8695751
  928859.4114904  811146.3700185  928856.2857064  811216.6827467
  928859.4114904   811376.056762  928873.4734216  811443.2447305
#Sta/Elev= 30
       0 2361.94   10.47 2358.05   16.92 2357.25   25.18  2357.2   50.19 2355.86
   59.65 2354.53   72.95 2346.59   77.18 2343.01  104.45  2336.4  159.51 2336.27
  175.77 2333.89  190.78 2331.57  196.54 2331.42  201.96 2331.79  208.22  2333.7
  213.67 2335.34  224.62 2336.19  249.67 2336.54  272.82 2337.92  299.26 2342.69
  310.52 2345.34  314.75 2346.89  358.68 2352.85   381.6 2356.78  386.59 2358.54
  390.49 2359.18  403.08 2363.91     420 2364.94  435.87 2365.19  441.75 2368.39
#Mann= 3 , 0 , 0
       0    .075       0  175.77     .05       0  208.22     .06       0
#XS Ineff= 2 , 0
       0  173.54 2336.42  219.54       0 2336.42
Permanent Ineff=
       F       F
#Block Obstruct= 2 ,-1
  276.18  313.522356.449    80.8  114.77 2358.25
Bank Sta=175.77,208.22
Exp/Cntr=0.5,0.3

Type RM Length L Ch R = 3 ,108398  ,,,
Node Photo=H:\PROJ\06-0741\CE\GIS\DATA\FRENCH_BROAD_RIVER\SHAPEFILES\survey_data\photos\FBSTR_1283.JPG
BEGIN DESCRIPTION:
108322  FBSTR_1283
END DESCRIPTION:
Bridge Culvert--1,0,-1,-1, 0
Deck Dist Width WeirC Skew NumUp NumDn MinLoCord MaxHiCord MaxSubmerge Is_Ogee
17,15,2.6,0, 7, 7, , , 0.95, 0, 1,1,,
       0  183.54  183.54  196.54  209.54  209.54  234.66
 2336.27 2336.42 2336.42 2336.42 2336.42 2336.42 2336.41
                 2335.42 2335.42 2335.42
       0     213     213  230.99     239     239  262.18
 2335.35 2336.42 2336.42 2336.42 2336.42 2336.42 2336.33
                 2335.42 2335.42 2335.42
BR Coef=-1 , 0 , 0 ,, 0 ,,,0.8,0,,0,
WSPro=,,,, 1 ,,,, 0 ,,,, 0 ,,,,-1 ,-1 ,-1 , 0 , 0 , 0 , 0 , 0
BC Design=,, 0 ,, 0 ,,,,,,

Type RM Length L Ch R = 1 ,108380  ,23.25,72.79,79.21
BEGIN DESCRIPTION:
108301.6
END DESCRIPTION:
XS GIS Cut Line= 6
  928900.0364402  810996.3692584   928864.098118  811038.5571002
  928845.3485351  811072.9325304  928814.0988888  811166.6824934
  928814.0988888  811311.9945775  928851.5990788  811436.9952109
#Sta/Elev= 30
       0 2363.01    4.94 2362.48   25.23 2357.34   53.46  2356.1   67.35 2354.95
   73.53  2353.7  101.27 2337.19  108.48 2336.01  143.59 2334.63  191.69 2335.35
  207.91 2333.61  222.99 2331.97  234.96 2331.81  238.292333.374  241.56 2334.91
  250.59  2335.6  263.04 2338.65  280.11 2338.34  318.92 2339.53  321.92 2339.18
  338.93 2341.91  357.45 2346.53     383 2350.57   410.2 2353.89  413.37 2354.77
  419.89 2355.53   430.3 2358.62  433.16 2361.07  447.03 2364.45  469.64 2365.27
#Mann= 3 , 0 , 0
       0    .065       0  207.91     .05       0  238.29     .06       0
#XS Ineff= 2 , 0
       0     203    2333     249       0    2333
Permanent Ineff=
       F       F
#Block Obstruct= 2 ,-1
  307.09  345.182353.587  103.64  132.542348.545
Bank Sta=207.91,238.29
Exp/Cntr=0.5,0.3

Type RM Length L Ch R = 1 ,108307  ,44.99,93.48,267.17
BEGIN DESCRIPTION:
108228.8
END DESCRIPTION:
XS GIS Cut Line= 6
  928851.5990788  811032.3075806   928771.911047   811135.431823
  928725.0365777  811221.3693743  928723.4736857  811293.2449946
  928765.6615275  811397.9321289   928771.911047  811469.8077491
#Sta/Elev= 30
       0 2355.07   15.18 2354.19   37.52 2344.33   43.58 2340.78    53.2 2336.72
   59.02 2334.71   75.73 2333.82   94.35 2333.57  105.03 2333.91  119.16 2335.19
  134.59 2334.95  157.17 2335.74  181.07 2333.15  194.15 2331.66  208.24 2331.11
  220.522332.875  240.04 2335.52   260.5 2335.33  279.99 2335.69  299.71 2336.71
  316.56 2338.05  362.84 2343.15  398.84  2347.7  411.97 2350.83  428.54 2360.26
  442.66 2365.23  458.07 2366.29  458.89 2367.38  480.97 2381.43  486.21 2381.75
#Mann= 3 , 0 , 0
       0     .07       0  181.07     .05       0  220.52     .06       0
#Block Obstruct= 2 ,-1
  312.12  330.912349.619   57.67   79.122346.581
Bank Sta=181.07,220.52
Exp/Cntr=0.3,0.1

Type RM Length L Ch R = 1 ,108213  ,92.8,293.09,390.05
BEGIN DESCRIPTION:
108135.3
END DESCRIPTION:
XS GIS Cut Line= 6
  928831.2855798  811030.7446887  928784.4111104  811046.3695118
  928629.7237227  811168.2443612  928585.9740131  811194.8073799
  928548.4738231   811210.432203  928476.5982029  811230.7446779
#Sta/Elev= 30
       0 2352.33    8.21 2351.98   19.12 2350.53   23.97 2348.63    37.7 2344.88
   47.65 2339.09   62.56 2332.87   79.28 2332.62   88.05 2331.45  101.06 2332.67
  132.91 2333.89  146.08 2333.57   164.1 2331.32  186.54 2329.72  201.58 2330.26
  208.75 2330.91  213.58 2331.27  221.97 2332.92  236.99 2335.17  245.66 2335.59
  281.03 2336.04  324.99 2335.07  351.44 2335.41  371.22 2338.44  373.04 2339.22
  379.39 2343.44  391.79 2352.88  402.74 2362.92  409.72 2368.58  413.05 2370.89
#Mann= 3 , 0 , 0
       0     .07       0   164.1     .05       0  208.75    .065       0
Bank Sta=164.1,208.75
Exp/Cntr=0.3,0.1

Type RM Length L Ch R = 1 ,107920  ,177.12,184.02,191.04
BEGIN DESCRIPTION:
107842.3
END DESCRIPTION:
XS GIS Cut Line= 4
  928848.4732949  810997.9321504  928776.5986988  810955.7443086
  928634.4113745   810876.057301  928556.2862347  810835.4323512
#Sta/Elev= 30
       0 2352.87   16.13 2350.47   31.89 2347.57   43.17 2345.73   46.99 2344.95
   55.59 2341.11   61.68 2338.53   66.51 2335.98   70.29 2334.51   75.57 2332.05
    98.7 2330.78  114.95 2330.34  121.93 2330.29  139.86 2329.86  149.08 2329.79
  179.57  2331.1  192.06 2331.23  205.01 2331.14  235.85 2326.81  249.32 2324.85
  250.63 2324.88   255.7 2324.36  256.78 2324.46  263.492326.651  268.15 2328.17
  269.75 2329.51  299.36 2350.37  319.56 2367.93     333 2378.31  334.39 2378.77
#Mann= 3 , 0 , 0
       0     .07       0  235.85     .05       0  263.49    .075       0
Bank Sta=235.85,263.49
Exp/Cntr=0.3,0.1

Type RM Length L Ch R = 1 ,107736  ,81.03,85.99,80.04
BEGIN DESCRIPTION:
107658.2
END DESCRIPTION:
XS GIS Cut Line= 4
  928878.1610733  810821.3693959  928812.5359968  810779.1825783
  928750.0356802  810733.8699767  928706.2859706  810699.4945465
#Sta/Elev= 30
       0 2367.32     .94 2366.87    2.02    2366   17.96 2356.87   21.75 2354.75
   24.58  2353.5   44.67  2340.6   51.72  2338.1   60.16 2334.07   68.02 2330.86
   82.37 2329.22   90.11 2327.86  108.67 2327.88  121.69 2327.75  133.96 2325.38
  141.37 2324.15  142.03 2323.94  147.08 2323.42  154.61 2322.29  162.16  2322.9
  166.05 2323.65  167.25 2323.89  169.48    2324  185.71 2331.04  188.28 2333.11
  191.96 2336.39   197.9 2341.26   203.6 2346.22  205.92 2348.03  210.85 2351.49
#Mann= 3 , 0 , 0
       0    .075       0  142.03     .05       0  166.05    .075       0
#Block Obstruct= 1 ,-1
   68.16   92.122343.849
Bank Sta=142.03,166.05
Exp/Cntr=0.5,0.3

Type RM Length L Ch R = 1 ,107650  ,51.85,48.97,42.83
BEGIN DESCRIPTION:
107572.2
END DESCRIPTION:
XS GIS Cut Line= 5
  928896.9106562  810741.6823883  928834.4113637  810694.8068947
  928809.4112371    810671.36966  928785.9740024  810652.6200771
   928734.410857  810632.3076022
#Sta/Elev= 27
       0 2352.21    1.68 2351.25   10.65 2346.54   24.83 2338.14   28.19 2336.26
   36.85 2334.05   45.28 2332.22   50.86 2331.33   65.94  2328.1   67.96 2327.99
   80.81 2327.81   83.98 2327.58   86.77 2327.74   95.16 2326.49  104.55 2323.86
  108.01 2323.17  110.01 2322.87  117.91 2322.78  119.76 2322.81  134.01 2324.64
   143.8 2325.88  153.53  2329.6  170.23 2339.95  174.85 2344.91  193.73 2364.68
  197.06 2368.45  197.83 2369.01
#Mann= 3 , 0 , 0
       0    .075       0  104.55     .05       0  134.01    .075       0
#XS Ineff= 2 , 0
       0   89.91 2333.28  145.91       0 2333.28
Permanent Ineff=
       F       F
#Block Obstruct= 1 ,-1
   34.37    66.62351.329
Bank Sta=104.55,134.01
Exp/Cntr=0.5,0.3

Type RM Length L Ch R = 3 ,107622  ,,,
Node Photo=H:\PROJ\06-0741\CE\GIS\DATA\FRENCH_BROAD_RIVER\SHAPEFILES\survey_data\photos\FBSTR_1773A.JPG
BEGIN DESCRIPTION:
107543  FBSTR_1773A
END DESCRIPTION:
Bridge Culvert--1,0,-1,-1, 0
Deck Dist Width WeirC Skew NumUp NumDn MinLoCord MaxHiCord MaxSubmerge Is_Ogee
25,10,2.6,0, 7, 7, , , 0.95, 0, 1,1,,
   40.64   99.91   99.91  117.91  135.91  135.91   159.3
 2333.23 2333.28 2333.28 2333.28 2333.28 2333.28 2333.18
                 2330.78 2330.78 2330.78
   47.68  102.86  102.86  120.86  138.86  138.86     174
 2333.19 2333.28 2333.28 2333.28 2333.28 2333.282332.457
                 2330.78 2330.78 2330.78
BR Coef=-1 , 0 , 0 ,, 0 ,,,0.8,0,,0,
WSPro=,,,, 1 ,,,, 0 ,,,, 0 ,,,,-1 ,-1 ,-1 , 0 , 0 , 0 , 0 , 0
BC Design=,, 0 ,, 0 ,,,,,,

Type RM Length L Ch R = 1 ,107601  ,130.45,96.67,44.6
BEGIN DESCRIPTION:
107523.3
END DESCRIPTION:
XS GIS Cut Line= 6
  928935.9737382  810699.4945465  928893.7858965  810674.4944198
  928846.9114271  810641.6818816  928814.0988888  810610.4322353
  928792.2235219  810605.7445835  928753.1614641  810604.1827157
#Sta/Elev= 29
       0 2356.02    1.15 2355.46   16.27 2349.56   22.87 2345.85   25.67 2344.77
   28.31 2343.54   37.72 2339.47   51.21 2330.92   54.45 2329.45   62.06 2327.98
   65.39  2327.6   79.93 2326.92   89.04 2326.87  105.86    2323  109.32 2322.72
  120.86 2322.25  136.05  2322.4  138.54 2322.71  143.41 2323.75  151.57 2325.48
  159.57 2327.93  171.26 2330.22  173.94 2332.41  177.94 2335.55  186.38 2341.92
  196.33 2348.27  200.63 2350.41  202.74 2351.23  213.03 2356.48
#Mann= 3 , 0 , 0
       0    .075       0  105.86     .05       0  143.41    .075       0
#XS Ineff= 2 , 0
       0   87.86    2330  153.86       0    2330
Permanent Ineff=
       F       F
#Block Obstruct= 1 ,-1
   45.87   77.562351.645
Bank Sta=105.86,143.41
Exp/Cntr=0.5,0.3

Type RM Length L Ch R = 1 ,107504  ,142.86,99.5,11.92
BEGIN DESCRIPTION:
107426.6
END DESCRIPTION:
XS GIS Cut Line= 6
  928982.8482076  810563.5567417  928882.8487251  810543.2442668
  928862.5362502  810533.8699875  928842.2237753  810536.9947472
  928798.4740657  810554.1824624  928737.5356168  810590.1197604
#Sta/Elev= 30
       0 2352.87    6.69 2348.29   11.41 2344.73   15.54  2341.4   29.42 2331.31
   32.57 2330.36   47.64 2325.31   61.13  2326.4   65.32 2326.64   67.95 2326.93
   91.11 2322.44   97.32  2321.1   114.5 2321.22   118.1 2321.33  121.79 2321.53
  125.69 2322.17  144.59 2323.95  156.25 2324.25  168.09 2325.47  179.09 2326.86
   184.9 2327.46   198.7 2330.29  204.92 2330.89  214.58 2336.65  216.95 2338.29
  237.19 2349.47  242.18    2352  252.31 2355.93  255.22 2357.53  262.74 2362.39
#Mann= 3 , 0 , 0
       0      .1       0   91.11     .05       0  125.69    .075       0
Bank Sta=91.11,125.69
Exp/Cntr=0.3,0.1

Type RM Length L Ch R = 1 ,107405  ,92.34,66.91,34.5
BEGIN DESCRIPTION:
107327.1
END DESCRIPTION:
XS GIS Cut Line= 6
  928945.3490418  810404.1827265   928901.598308  810435.4323727
  928851.5990788  810469.8067788  928803.1606933  810507.3069688
  928770.3481551  810560.4319819   928734.410857  810580.7444568
#Sta/Elev= 30
       0 2361.05    6.85  2355.9   13.62 2349.43   23.17 2340.96   28.62 2334.95
   33.02 2330.84   40.88 2325.69    48.3 2322.67   55.27 2320.98   59.54 2320.18
   82.15 2320.64   94.56 2320.53    99.9 2320.24  107.65 2320.29  120.45 2322.46
  130.95 2323.05  136.11 2323.59  149.98 2323.73   182.8 2323.23  198.13 2325.09
  207.14 2326.73  216.59  2328.8  221.89 2330.25  223.77 2330.47  227.35 2332.19
  248.21 2343.98  261.57 2353.16  270.74 2356.85  272.82 2357.38  279.42 2360.25
#Mann= 3 , 0 , 0
       0    .095       0   55.27     .05       0   82.15    .075       0
Bank Sta=55.27,82.15
Exp/Cntr=0.3,0.1

Type RM Length L Ch R = 1 ,107338  ,182.59,159.16,35.4
BEGIN DESCRIPTION:
107260.2
END DESCRIPTION:
XS GIS Cut Line= 6
  928839.0990155  810361.9948847  928831.2855798  810410.4322461
  928818.7865406  810452.6200878  928803.1606933  810476.0573225
  928723.4736857  810569.8072855  928695.3487992  810604.1827157
#Sta/Elev= 30
       0 2358.06     6.9 2352.67    17.2 2342.36   27.71 2333.05   29.87 2330.87
   41.86 2324.98   58.52 2320.64   61.94 2319.69   68.16 2318.96   73.24 2318.95
   81.41 2319.56   88.85 2320.56  113.27 2323.21   127.8 2323.24  160.03 2322.51
  165.05 2322.59   182.3 2324.22  186.62 2325.35  201.31 2327.92  207.41  2329.8
  211.18 2332.15  226.25  2340.9  237.11 2347.89  238.89 2348.66  244.13 2351.94
  265.39 2363.78  271.71 2365.26  277.16 2369.89  283.28 2371.81  288.71 2371.59
#Mann= 3 , 0 , 0
       0    .095       0   58.52     .05       0   88.85    .075       0
Bank Sta=58.52,88.85
Exp/Cntr=0.3,0.1
