HEC-RAS study lds_big_laurel_crk.prj: lds_big_laurel_crk

--- lds_big_laurel_crk.g20 (geometry) --- (continued)

Type RM Length L Ch R = 1 ,76108   ,242.77,281.12,288.79
BEGIN DESCRIPTION:
76030.53
END DESCRIPTION:
XS GIS Cut Line= 4
  913940.6611735  809588.5569222  914026.5987248  809652.6201309
   914078.160846  809696.3698405  914128.1610994  809741.6824421
#Sta/Elev= 30
       0 2005.03    7.65  2004.5   11.72 2003.63   21.61 1996.95   29.17 1992.83
   32.28 1990.61   40.99 1980.36   42.95 1978.27   55.69 1971.89   59.27 1971.32
   69.54 1970.55   81.01 1970.21   87.85 1969.55   97.03 1966.87  102.97 1966.12
  107.69 1964.74   110.1  1964.7  126.14 1961.63  136.99 1960.26  144.62 1958.94
  150.81 1958.14  154.63 1957.94  180.49 1957.16  182.26 1957.26  183.761958.494
  210.16 1979.64  221.32 1986.13  222.84 1987.16   232.8  1995.5  242.29  2005.8
#Mann= 3 , 0 , 0
       0    .075       0  154.63     .05       0  183.76    .075       0
Bank Sta=154.63,183.76
Exp/Cntr=0.3,0.1

Type RM Length L Ch R = 1 ,75827   ,96.57,113.63,145.34
BEGIN DESCRIPTION:
75749.41
END DESCRIPTION:
XS GIS Cut Line= 5
  913779.7232421  809735.4318983  913804.7233687  809785.4321517
  913831.2863874  809838.5571648  913892.2238121  809911.9946529
  913907.8486352  809954.1824947
#Sta/Elev= 30
       0 1999.35    9.22 1996.54   21.25 1994.26   26.71 1992.53   29.18 1991.16
   52.15 1976.56      61 1970.57   67.01 1967.84   75.66 1968.32   85.58 1967.83
  101.56 1960.91  106.82 1958.07  108.49 1957.31   115.3 1956.61  117.38 1956.25
  134.52 1955.41  147.62 1956.13  149.98 1956.38  160.85 1958.43  166.11  1959.4
  184.33 1962.38   193.6 1963.54  200.23 1965.25  210.62 1967.53  218.24 1970.34
  223.95 1972.14  232.91 1975.31  240.07 1979.57  253.65 1991.15  255.71 1993.08
#Mann= 3 , 0 , 0
       0    .075       0  108.49     .05       0  160.85     .07       0
Bank Sta=108.49,160.85
Exp/Cntr=0.3,0.1

Type RM Length L Ch R = 1 ,75714   ,72.58,130.08,137.76
BEGIN DESCRIPTION:
75635.78
END DESCRIPTION:
XS GIS Cut Line= 5
  913710.9734058  809752.6196135  913712.5362978  809808.8693864
  913735.9735325  809883.8697664  913756.2860074  809957.3072545
  913756.2860074  809994.8074445
#Sta/Elev= 30
       0 2001.44    2.02 2000.67    7.28 1998.98   22.44 1993.58    33.1 1990.26
   37.38 1988.35   43.51 1987.21   55.63 1978.04   67.08 1968.72   71.39 1965.88
   72.39 1965.67   77.83 1965.04   81.73 1965.19   87.43 1965.59   98.42 1965.17
  109.32    1962   119.6 1958.61   130.1 1956.04  149.73 1954.76  165.68 1954.76
   174.4 1955.99   179.2 1956.54  184.32  1957.7  195.16 1963.31  211.04 1983.39
  212.53 1985.21  218.45 1989.51  229.22 1997.17  245.05 2006.87  248.54 2010.14
#Mann= 3 , 0 , 0
       0    .075       0   130.1     .05       0   179.2     .07       0
Bank Sta=130.1,179.2
Exp/Cntr=0.3,0.1

Type RM Length L Ch R = 1 ,75584   ,101.7,150.52,205.55
BEGIN DESCRIPTION:
75505.70
END DESCRIPTION:
XS GIS Cut Line= 6
  913654.7236328   809760.432025  913635.9740499  809826.0571015
  913617.2234428  809883.8697664  913610.9739233  809918.2451966
   913615.661575  809944.8071911  913626.5987464  809990.1197927
#Sta/Elev= 28
       0 1994.62   22.93 1984.62      27 1983.33    29.5 1982.22   42.78 1977.36
   50.14 1974.04   54.47 1972.36   67.37  1963.2   69.85 1963.63   75.54 1963.74
   81.46 1963.31    86.2 1963.21   94.65 1963.27  101.95 1961.25  113.36 1958.33
  123.01 1957.03  127.82  1956.5  135.98 1955.93  143.69 1954.92  150.56 1953.72
  159.75 1953.93  166.62 1953.76  172.47 1953.84  184.71 1954.53  188.84 1959.53
  194.13 1967.79  218.45 1994.01  237.55 2015.89
#Mann= 3 , 0 , 0
       0     .08       0  135.98     .05       0  188.84     .07       0
Bank Sta=135.98,188.84
Exp/Cntr=0.5,0.3

Type RM Length L Ch R = 1 ,75433   ,67.33,62.85,115.28
BEGIN DESCRIPTION:
75355.17
END DESCRIPTION:
XS GIS Cut Line= 6
   913556.425306   809753.765666  913530.3528675  809800.8644298
  913519.4187686  809814.7420093  913418.9133434  809890.4367804
  913403.7739795  809919.4526997  913402.0922831  809936.6946961
#Sta/Elev= 30
       0 1980.62    5.99 1978.38    8.36 1977.73    19.3 1973.39   29.27 1969.61
    45.6 1963.01   52.21 1961.76   60.02  1960.8   75.65 1961.13   82.03 1961.17
   86.71 1961.37    90.1 1960.83   94.46 1961.39   99.88 1961.51  107.16 1956.57
  108.93 1955.37  112.77  1953.1  139.87 1952.79  146.91 1954.28  150.62  1954.9
  151.32    1955  171.54  1962.8  174.39 1963.71  178.29 1966.92  185.63 1973.89
  197.67 1981.11  208.18 1987.87  214.54 1991.09  233.03 1997.76  247.77 2004.71
#Mann= 3 , 0 , 0
       0     .09       0  107.16     .05       0  150.62     .07       0
#XS Ineff= 2 , 0
       0     105  1962.5               0
Permanent Ineff=
       F       F
Bank Sta=107.16,150.62
Exp/Cntr=0.5,0.3

Type RM Length L Ch R = 3 ,75400   ,,,
BEGIN DESCRIPTION:
75321  FBSTR_1277  No Photo
END DESCRIPTION:
Bridge Culvert--1,0,-1,-1, 0
Deck Dist Width WeirC Skew NumUp NumDn MinLoCord MaxHiCord MaxSubmerge Is_Ogee
18,32,2.6,0, 4, 5, , , 0.95, 0, 0,0,,
   96.46     105     140     175
 1961.39  1962.8  1962.8  1962.8
          1960.8  1960.8  1960.8
   70.13     106     141     176  184.31
 1961.35  1962.8  1962.8  1962.8 1960.78
          1960.8  1960.8  1960.8
BR Coef=-1 , 0 , 0 ,, 0 ,,,0.8,0,,0,
WSPro=,,,, 1 ,,,, 0 ,,,, 0 ,,,,-1 ,-1 ,-1 , 0 , 0 , 0 , 0 , 0
BC Design=,, 0 ,, 0 ,,,,,,

Type RM Length L Ch R = 1 ,75370   ,109.15,106.68,20.85
BEGIN DESCRIPTION:
75292.33
END DESCRIPTION:
XS GIS Cut Line= 6
  913510.5883265  809703.7223972  913486.6185205  809748.7185285
  913427.3238735  809808.8540237  913331.8645614  809822.7316033
   913322.612159  809863.5224695  913345.3212048  809924.9197491
#Sta/Elev= 30
       0 1995.46   13.83 1988.66   21.07  1985.8   35.59 1978.42    45.9 1974.11
   58.07  1968.1   70.13 1961.35   88.67 1957.31   96.49 1955.15  108.68 1953.96
   127.9 1952.95  135.32 1953.18  145.19 1956.58  159.24 1959.92  170.76 1961.21
  201.08  1960.6  213.69 1960.79  215.92 1961.51  220.44  1961.2  226.93 1961.35
   233.1 1963.28  240.07 1966.34  254.68 1973.83  280.31 1980.47  289.32 1984.73
  296.45 1985.54  314.43 1993.11   317.3 1994.07   335.9 1997.79  341.74 1999.92
#Mann= 3 , 0 , 0
       0    .095       0   96.49     .05       0  145.19     .06       0
#XS Ineff= 2 , 0
       0   87.35  1957.6     176       0 1961.14
Permanent Ineff=
       F       F
Bank Sta=96.49,145.19
Exp/Cntr=0.5,0.3

Type RM Length L Ch R = 1 ,75264   ,314.14,295.17,241.64
BEGIN DESCRIPTION:
75185.65
END DESCRIPTION:
XS GIS Cut Line= 6
  913412.5358018  809672.9326058  913348.4736173  809738.5576823
  913329.7240344   809761.994917  913310.9734273  809785.4321517
  913310.9734273   809835.432405  913314.0981871  809915.1194127
#Sta/Elev= 30
       0 1983.98    2.58 1982.88     7.4 1980.48   21.12 1974.49   28.83 1970.04
   35.27 1967.31   42.22 1963.52   57.99  1954.1   67.47 1953.07   75.39  1950.4
   84.45 1950.71   96.88 1951.44  104.73 1953.99  109.34 1955.74  111.23 1955.92
  117.31 1957.09  128.11 1959.61  143.71 1959.92  158.08 1959.97  173.44 1960.41
  186.43 1965.66  202.66 1971.61  216.32 1974.78  218.49 1975.49  235.85 1980.09
  244.45 1982.19  252.95 1984.81  263.15 1988.58  273.52 1991.64  281.49 1994.16
#Mann= 3 , 0 , 0
       0     .09       0   67.47     .05       0  104.73     .07       0
Bank Sta=67.47,104.73
Exp/Cntr=0.3,0.1

Type RM Length L Ch R = 1 ,74968   ,205.85,164.27,31.51
BEGIN DESCRIPTION:
74890.49
END DESCRIPTION:
XS GIS Cut Line= 5
  913129.7240452  809515.1194342  913103.1610265  809574.4949911
  913089.0980712  809615.1199409  913081.2856596  809657.3067585
  913085.9733114  809776.0568481
#Sta/Elev= 30
       0  2007.2    2.42 2005.17   13.71 1994.47   41.72 1962.07      52 1952.52
   54.281951.266   58.42 1948.99   63.74 1948.16   82.28  1948.9   92.32 1950.03
   95.37 1950.68  107.46 1953.41  120.45 1954.29  136.83 1955.13  157.12 1956.64
  159.47 1956.83  169.22 1958.14  171.11 1958.54  173.86 1959.63  186.24 1963.46
  196.57 1965.88  201.22 1965.92  213.98 1965.66  230.01 1969.88   244.3 1974.11
  246.43 1974.42  251.75 1975.99  256.77 1976.75  265.45 1977.53  269.78 1978.41
#Mann= 3 , 0 , 0
       0      .1       0   54.28     .05       0   95.37    .065       0
Bank Sta=54.28,95.37
Exp/Cntr=0.3,0.1

Type RM Length L Ch R = 1 ,74804   ,176.07,143.65,76.19
BEGIN DESCRIPTION:
74726.21
END DESCRIPTION:
XS GIS Cut Line= 6
  912912.5363408  809538.5576931  912950.0365309  809622.9323525
  912989.0985887  809651.0572389  913020.3482349  809682.3068852
  913048.4731214   809722.931835  913065.6608365  809782.3073919
#Sta/Elev= 30
       0 1995.44    3.43 1991.69    7.16  1986.3    8.64 1983.86   29.43 1959.01
   36.831949.856   38.66  1947.6   39.49 1946.97   50.32  1947.7   53.44 1947.39
    78.9  1949.9  120.68  1952.5  137.29 1953.39   148.5 1954.31   156.5 1954.71
  170.86 1956.37  180.09 1957.28  186.28 1957.69  193.64 1958.68  207.52 1964.03
  211.93 1965.45  218.38 1967.91  224.22  1967.8  231.95 1967.42  243.09 1966.44
  261.87 1973.98  267.21 1974.85   273.6 1975.74  281.19  1976.6  295.95 1978.78
#Mann= 3 , 0 , 0
       0     .08       0   36.83     .05       0    78.9    .065       0
Bank Sta=36.83,78.9
Exp/Cntr=0.3,0.1

Type RM Length L Ch R = 1 ,74660   ,272.71,268.09,254.7
BEGIN DESCRIPTION:
74582.57
END DESCRIPTION:
XS GIS Cut Line= 6
  912790.6614914   809688.557429  912853.1607839  809715.1194234
  912895.3486257  809727.6194868    913000.03576  809777.6197401
  913042.2236018  809819.8075819  913054.7236652  809847.9324684
#Sta/Elev= 30
       0  2001.3   14.04 1989.88   27.84 1976.83   37.51 1965.86   44.27 1962.21
    54.7 1955.45   56.96 1954.26   58.05 1953.07   64.35  1950.3   69.36 1947.99
   79.93 1947.18   97.72 1947.65  111.91 1948.85  130.82 1950.38  135.14 1950.47
  138.92 1951.95  160.51 1957.23   179.8 1959.24  193.44 1961.27  199.75 1963.69
  203.28  1965.5  215.84 1970.26   221.7 1969.78  229.64 1969.82  236.12 1970.69
  254.52 1978.23  261.16 1978.35  267.58 1979.27  281.85 1980.64  318.38 1985.93
#Mann= 3 , 0 , 0
       0    .075       0   64.35     .05       0  111.91     .06       0
Bank Sta=64.35,111.91
Exp/Cntr=0.3,0.1

Type RM Length L Ch R = 1 ,74392   ,325.54,304.29,311.15
BEGIN DESCRIPTION:
74314.48
END DESCRIPTION:
XS GIS Cut Line= 4
  912690.6609847  809938.5576715  912735.9735863  809960.4320142
  912900.0362775  810007.3075078    913000.03576  810049.4943254
#Sta/Elev= 30
       0    1983    8.38 1979.02    16.9 1972.89   37.01 1960.57   42.34 1957.75
   47.53 1953.09   50.09    1952    62.8 1949.61   79.76 1948.57   92.81 1945.78
  106.57 1944.19   133.6 1945.03  137.38 1946.02  144.14 1947.55  166.51 1954.11
     179 1955.13  188.21 1957.44  202.21 1960.11  215.86 1965.71  237.59 1972.11
  247.03 1975.79  254.98 1979.95  271.17 1983.33  279.18 1983.16  285.11 1983.75
  292.95 1992.33  295.79 1992.59  299.32 1994.07  306.56 1994.23  329.48 1998.23
#Mann= 3 , 0 , 0
       0    .075       0   92.81     .05       0  137.38    .065       0
Bank Sta=92.81,137.38
Exp/Cntr=0.3,0.1

Type RM Length L Ch R = 1 ,74088   ,58.93,174.42,264.08
BEGIN DESCRIPTION:
74010.19
END DESCRIPTION:
XS GIS Cut Line= 5
  912511.9013735  810207.0821784  912596.2760329  810250.8329122
  912679.0888245  810260.2071915   912782.214091    810289.89497
  912840.0267559  810339.8952233
#Sta/Elev= 30
       0 1976.97    6.45 1976.09   16.92 1973.46   27.52 1971.69   39.31 1967.35
   44.51 1965.85   54.76 1963.85   69.71 1958.51   80.94  1955.9   95.04 1951.51
  107.13 1950.02  118.33 1950.75  134.33 1950.87  141.51 1949.38  155.741943.609
  160.79  1941.6  176.93 1942.58  195.01 1942.89  208.84 1944.02   239.1 1947.81
  256.23 1950.92  269.64 1954.52  283.49 1959.48  296.29 1966.92  305.33 1973.25
  314.88 1980.36  331.92 1995.23   339.5 2000.17   350.8 2002.85  362.13 2003.16
#Mann= 3 , 0 , 0
       0    .075       0  155.74     .05       0  208.84    .065       0
Bank Sta=155.74,208.84
Exp/Cntr=0.3,0.1

Type RM Length L Ch R = 1 ,73914   ,163.13,248.31,253.66
BEGIN DESCRIPTION:
73835.76
END DESCRIPTION:
XS GIS Cut Line= 6
  912496.2765504  810232.0823051  912549.4015635  810302.3950333
  912585.3388615  810346.1447429  912596.2760329  810394.5831285
    912615.02664  810422.7080149  912605.6513364   810496.145503
#Sta/Elev= 30
       0 1975.42    7.95 1973.58   14.09 1972.36   20.48 1970.84   44.45  1963.6
   47.55 1962.78   52.07 1961.41   59.46 1958.52   73.87 1954.28   88.13 1951.55
   96.61 1950.67   106.8 1949.75  110.38 1949.61  118.18 1949.35  131.27 1949.19
  144.74 1949.48  157.01 1948.39  168.55 1946.72  197.53  1942.3  206.66 1941.11
  215.33 1939.62   216.6 1939.56   228.2 1940.32  234.37 1940.39  240.19 1940.23
  248.22 1940.28  252.181943.347  286.31 1969.51  297.94 1978.07  302.24 1980.71
#Mann= 3 , 0 , 0
       0    .075       0  197.53     .05       0  252.18    .075       0
Bank Sta=197.53,252.18
Exp/Cntr=0.3,0.1

Type RM Length L Ch R = 1 ,73665   ,366.73,436.46,474.39
BEGIN DESCRIPTION:
73587.46
END DESCRIPTION:
XS GIS Cut Line= 6
  912388.4636321  810263.3329755   912372.838809  810352.3952867
  912369.7140492  810386.7696927  912358.7758536   810419.582231
  912355.6510939  810444.5823577  912355.6510939  810508.6455663
#Sta/Elev= 29
       0 1972.05     5.5 1970.44   10.78 1969.05   14.42 1968.21   24.05 1965.18
   41.95  1959.8   57.31 1955.68   70.02 1950.97   77.79 1948.41   84.99 1945.71
   87.04 1945.27   97.96 1943.38  124.94  1940.5  139.74 1939.07   154.4 1939.26
  162.22 1939.44  168.31 1939.31  171.99 1939.99  179.22 1940.44  183.39  1941.2
  184.72 1941.54  193.08 1943.68  196.11 1944.67  202.03 1947.67  211.41 1953.04
  224.59 1962.09  230.06    1966  239.24 1972.99  248.78 1978.69
#Mann= 3 , 0 , 0
       0    .075       0  124.94     .05       0  184.72    .075       0
Bank Sta=124.94,184.72
Exp/Cntr=0.3,0.1

Type RM Length L Ch R = 1 ,73229   ,488.27,445.16,421.63
BEGIN DESCRIPTION:
73151
END DESCRIPTION:
XS GIS Cut Line= 6
  912079.0888568   810161.770601   912036.901015  810205.5203106
  911977.5264823  810247.7071282  911940.0262923  810288.3331022
  911922.8385772  810310.2074449   911905.650862  810346.1447429
#Sta/Elev= 30
       0 1959.79     8.7 1958.64   13.85 1957.72   18.67 1957.34   31.83  1954.9
   34.79 1954.62   38.73    1954    42.7 1953.53   71.63 1949.24   76.64  1948.7
  100.61 1945.25  105.01  1944.7  110.43 1943.74  117.26 1942.18  131.22 1938.56
  133.19 1938.13  138.12 1937.61   143.8 1936.66  165.18  1936.9  172.96    1939
  212.59 1952.68  215.85 1954.48  219.67 1957.06  226.65 1962.21  229.07 1963.66
   233.7 1967.12   242.6 1973.28  249.97  1977.6  253.36 1980.05  256.56  1981.8
#Mann= 3 , 0 , 0
       0     .07       0  131.22     .05       0  172.96     .07       0
Bank Sta=131.22,172.96
Exp/Cntr=0.3,0.1

Type RM Length L Ch R = 1 ,72784   ,219.32,209.77,219.32
BEGIN DESCRIPTION:
72705.83
END DESCRIPTION:
XS GIS Cut Line= 4
  911599.4008465   809991.457366   911574.401744  810050.8329229
  911544.7139656   810121.144627  911516.5890791  810224.2698935
#Sta/Elev= 23
       0 1970.36   21.86 1954.33   22.65 1953.88    37.5  1948.7   50.32 1942.24
   67.041934.295   69.24 1933.25   86.88 1932.96   90.58 1932.68   100.6 1933.01
  114.36 1934.32  120.13 1936.85  128.72 1940.61  134.25 1941.79  143.08  1943.3
  149.06 1944.43  157.58 1946.22  172.18 1949.79  186.61 1953.86  201.56 1958.81
  215.17 1962.71  242.82 1970.11  247.64 1971.48
#Mann= 3 , 0 , 0
       0     .09       0   67.04     .05       0  120.13    .055       0
Bank Sta=67.04,120.13
Exp/Cntr=0.3,0.1

Type RM Length L Ch R = 1 ,72574   ,84.79,112.49,133.67
BEGIN DESCRIPTION:
72496.06
END DESCRIPTION:
XS GIS Cut Line= 5
  911405.6514011  809905.5198147  911383.7760342  809950.8324162
   911368.151211  810005.5203214  911340.0263246  810068.0206381
  911304.0890265  810127.3951708
#Sta/Elev= 22
       0 1971.31    4.18 1971.13   37.26 1955.53   50.32 1948.79   80.781932.766
   83.68 1931.24      91 1931.34    93.5 1931.19   95.33 1931.49  110.04 1932.89
  118.15 1934.49   126.5 1936.95  133.82 1938.26  138.28 1939.27  152.46 1940.47
  166.46 1942.29  197.48 1946.64  211.76  1948.5   216.1 1950.08  230.58 1955.79
  234.75 1957.62  245.13 1960.32
#Mann= 3 , 0 , 0
       0     .08       0   80.78     .05       0  118.15     .07       0
Bank Sta=80.78,118.15
Exp/Cntr=0.3,0.1

Type RM Length L Ch R = 1 ,72462   ,81.54,103.23,152.88
BEGIN DESCRIPTION:
72383.57
END DESCRIPTION:
XS GIS Cut Line= 6
  911363.4635593  809885.2073398  911305.6508943  809921.1446378
  911279.0888999  809943.0200047  911254.0887732  809968.0201314
  911210.3390636  810025.8327963  911177.5265254   810047.707139
#Sta/Elev= 27
       0  1969.5    3.53 1968.24   16.76 1962.18   47.57 1948.68   68.07 1941.63
   80.55 1937.24   89.83 1933.87    93.31932.525   95.91 1931.56      97 1931.41
   104.4 1931.47   122.5 1931.39  124.01 1931.39  126.59 1931.73  137.84 1932.71
  145.91 1933.59  164.61 1938.88   171.9 1941.07  186.51 1947.68  187.29  1948.1
  194.44 1951.04  210.39 1957.85  216.83 1960.75  225.03 1962.92  236.66 1966.14
   242.2 1968.68  249.83 1971.17
#Mann= 3 , 0 , 0
       0    .075       0    93.3     .05       0  137.84    .075       0
Bank Sta=93.3,137.84
Exp/Cntr=0.3,0.1

Type RM Length L Ch R = 1 ,72358   ,325.51,397.01,415.57
BEGIN DESCRIPTION:
72280.35
END DESCRIPTION:
XS GIS Cut Line= 6
   911333.776805  809839.8947382  911297.8384828  809839.8947382
  911268.1517285  809847.7071497  911227.5267787  809864.8948649
  911141.5892273  809888.3331237  911118.1509685  809888.3331237
#Sta/Elev= 27
       0 1958.59   26.92 1945.51   37.33  1943.3    38.1 1943.04   39.15 1942.85
   52.77 1941.31   54.76 1940.76   64.46  1937.2   87.35 1932.31   88.88 1931.85
   92.96  1931.5   98.53 1931.65  110.75 1930.92  117.02 1930.65  122.53 1930.41
  130.82 1929.69  135.99 1929.67  145.19 1929.93  146.63  1930.9  158.97 1935.97
  165.33 1940.87  172.34 1946.38  188.67 1961.43  192.84 1964.55  200.87 1969.18
  212.33 1975.35  223.36 1981.68
#Mann= 3 , 0 , 0
       0     .07       0  117.02     .05       0  146.63    .075       0
Bank Sta=117.02,146.63
Exp/Cntr=0.3,0.1

Type RM Length L Ch R = 1 ,71961   ,302.02,242.23,213.57
BEGIN DESCRIPTION:
71883.34
END DESCRIPTION:
XS GIS Cut Line= 6
  911321.2767417  809489.8950131  911279.0888999  809514.8951397
  911238.4639501  809525.8323111  911199.4008681  809525.8323111
  911077.5260186  809496.1455568  910990.0265995  809491.4579051
#Sta/Elev= 30
       0 1951.31   18.16 1948.66   22.47 1947.93    39.5 1945.77   49.04 1944.23
   58.74  1942.9   70.97 1940.88   79.93 1938.96   87.13 1937.92   94.17 1937.26
  100.89 1936.25  106.91 1935.64  112.47 1935.13  150.05 1933.05  169.76 1932.28
   182.3 1931.85  190.09  1931.7  207.74 1931.63  213.14 1931.82  223.52 1929.38
  230.89 1927.44  242.36 1927.45  251.02 1926.94  269.46  1929.6  288.58 1945.57
  315.06 1967.93  319.32 1971.67   325.6 1976.95  330.81 1980.47  343.29 1989.87
#Mann= 3 , 0 , 0
       0     .05       0  223.52     .05       0  269.46    .075       0
Bank Sta=223.52,269.46
Exp/Cntr=0.3,0.1

Type RM Length L Ch R = 1 ,71719   ,142.72,107.69,88.07
BEGIN DESCRIPTION:
71641.11
END DESCRIPTION:
XS GIS Cut Line= 6
  911227.5267787  809205.5203644  911171.2759816  809241.4576625
  911141.5892273   809250.832966  911060.3383035  809266.4577891
  911032.2134171  809278.9578525  910971.2759924  809318.0199103
#Sta/Elev= 29
       0 1967.08    4.82 1965.14   33.39 1950.07   42.45 1944.94   50.22 1940.65
   63.86 1935.73    69.7 1933.86   82.16 1928.65   90.61 1927.49   95.15 1928.72
  101.25  1929.5  113.66 1929.38  122.34 1929.48  132.26 1928.89  132.78 1928.78
  149.29 1924.93  155.37 1924.69  158.55 1925.04  165.09    1926   171.8 1926.02
  179.88 1926.83  183.43 1927.01  194.17 1928.91  208.89 1937.77  249.11 1959.43
   254.5 1961.85  259.76 1963.39  280.87 1970.44  283.83 1971.18
#Mann= 3 , 0 , 0
       0     .08       0  132.78     .05       0   171.8     .07       0
Bank Sta=132.78,171.8
Exp/Cntr=0.3,0.1

Type RM Length L Ch R = 1 ,71611   ,86.28,63.07,34.21
BEGIN DESCRIPTION:
71533.42
END DESCRIPTION:
XS GIS Cut Line= 6
   911129.089164  809094.5826864  911077.5260186  809136.7705282
  910980.6512959  809203.9574725   910961.901713  809222.7080795
  910950.9635175  809255.5206178  910949.4016497  809283.6455043
#Sta/Elev= 21
       0  1972.8    1.61  1971.5   13.83 1960.63   23.32 1955.48   43.56 1942.16
   48.89    1940   80.66  1925.6   83.11 1924.43   84.12  1924.3  106.83 1923.53
  114.28 1923.55  116.42 1923.81  129.66 1925.94  173.47 1932.62  183.63 1934.88
  189.34  1938.6  196.35  1939.3  208.74 1944.71  211.15 1945.45  249.84 1959.74
  273.91 1968.16
#Mann= 3 , 0 , 0
       0     .08       0   80.66     .05       0  129.66    .075       0
Bank Sta=80.66,129.66
Exp/Cntr=0.3,0.1

Type RM Length L Ch R = 1 ,71548   ,191.75,151.03,41.16
BEGIN DESCRIPTION:
71470.35
END DESCRIPTION:
XS GIS Cut Line= 6
  911065.0259553  809024.2699581  911036.9010688  809060.2072562
  911021.2762457  809096.1455784  910957.2140612  809149.2705915
  910932.2139345  809225.8328393  910932.2139345  809269.5825489
#Sta/Elev= 24
       0 1984.13   46.79 1942.81   53.81 1937.69   64.53 1931.28   67.04  1929.7
   77.26 1926.04      84 1923.72  101.08 1922.53  103.33 1922.58  108.93 1923.34
  118.53 1925.61  120.88 1925.99  164.25 1934.28  166.94 1934.68   196.8 1933.94
  203.02 1934.44  207.31 1934.69  220.78 1938.79  226.16  1940.7  235.37 1944.94
  249.22 1949.25  269.96 1955.36  281.57 1959.74  292.97 1963.71
#Mann= 3 , 0 , 0
       0     .08       0   77.26     .05       0  118.53    .075       0
Bank Sta=77.26,118.53
Exp/Cntr=0.3,0.1

Type RM Length L Ch R = 1 ,71397   ,58.42,81.5,113.7
BEGIN DESCRIPTION:
71319.32
END DESCRIPTION:
XS GIS Cut Line= 6
  910857.2135545  809041.4576732  910857.2135545  809086.7702748
  910875.9641616  809132.0828764  910900.9642883  809171.1449342
  910900.9642883  809194.5821689  910911.9014596  809264.8948972
#Sta/Elev= 29
       0 1971.53   12.39 1961.05   13.91 1960.16   28.16 1949.87    33.7 1946.25
   45.31 1937.78   50.64 1934.05    57.3 1930.08   71.55 1925.61   78.17 1923.14
   86.36 1922.91   92.36  1922.9   94.36 1922.94   98.88 1924.34  100.971924.672
  109.77 1926.07  120.28 1926.17   138.1 1931.49  140.94 1932.17  146.24 1933.61
  152.77 1935.19  154.45 1935.69  164.37 1938.97  171.91  1941.6  177.66  1942.9
  206.71 1951.15  221.63 1956.15  226.74  1957.6  235.53 1960.62
#Mann= 3 , 0 , 0
       0    .095       0   71.55     .05       0  100.97     .07       0
Bank Sta=71.55,100.97
Exp/Cntr=0.3,0.1

Type RM Length L Ch R = 1 ,71316   ,237.49,252.22,258.13
BEGIN DESCRIPTION:
71237.82
END DESCRIPTION:
XS GIS Cut Line= 6
    910830.65156  809028.9576099  910800.9637816  809075.8331035
   910794.714262  809107.0827497   910794.714262  809160.2077629
  910785.3389585  809180.5202378  910760.3388318  809227.3947071
#Sta/Elev= 21
       0 1975.42    5.75 1971.53     8.5 1969.24   13.92 1966.35   26.65 1957.54
   60.07 1933.65   69.66 1927.75   77.48 1925.53   82.57 1924.31   87.35 1923.94
  101.46 1922.16  118.36 1922.29  123.56 1922.59  129.54 1922.48  131.261923.581
   140.4 1929.43  159.63  1941.5  174.81 1952.77  179.62 1955.95  198.76 1964.87
  215.98 1973.43
#Mann= 3 , 0 , 0
       0      .1       0   87.35     .05       0  131.26    .075       0
Bank Sta=87.35,131.26
Exp/Cntr=0.3,0.1

Type RM Length L Ch R = 1 ,71064   ,456.9,412.62,314.09
BEGIN DESCRIPTION:
70985.60
END DESCRIPTION:
XS GIS Cut Line= 4
  910610.3390959  808938.3324067  910565.0264943  809021.1451983
  910546.2758872  809074.2702115  910536.9016079  809146.1448075
#Sta/Elev= 24
       0 1963.26   11.87 1955.83    20.5  1949.8    33.7 1942.65   56.95 1931.65
   66.42 1928.42    94.4    1923   98.49 1922.23  101.44  1921.7  101.91 1921.73
  105.09 1921.18  114.67 1919.52  116.01 1919.37  129.11 1919.87  129.47 1919.89
  130.19 1919.88  132.88    1921  143.95 1925.61  150.74 1926.41  153.83 1926.88
  166.27 1928.31  201.76 1952.59  216.31 1961.45  223.22 1965.12
#Mann= 3 , 0 , 0
       0      .1       0  105.09     .05       0  132.88    .075       0
Bank Sta=105.09,132.88
Exp/Cntr=0.3,0.1

Type RM Length L Ch R = 1 ,70651   ,277.05,221.53,79.59
BEGIN DESCRIPTION:
70572.98
END DESCRIPTION:
XS GIS Cut Line= 6
  910165.0265159  808855.5206393  910169.7141676  808938.3324067
   910180.651339  808982.0831405  910202.5267059  809025.8328501
  910243.1516557  809086.7702748  910277.5260617  809152.3953513
#Sta/Elev= 30
       0 1956.76   33.49 1934.93   46.61 1924.75   50.43 1921.22    53.7 1919.67
   56.34  1918.7    58.7 1917.84    67.9 1917.94   83.95 1918.55  102.76 1921.22
  133.28 1924.92  148.92 1925.51  161.93 1926.57  175.38 1927.95  183.89 1928.51
  194.06 1929.51  200.12  1929.1  207.53 1929.24  218.57 1929.16  229.28 1929.45
  245.55 1931.81  249.88 1932.28  262.38 1936.43   268.6 1938.19  289.64 1945.79
  292.23  1946.9  299.23 1949.53  306.31 1951.57  309.79 1953.02  324.28 1957.89
#Mann= 3 , 0 , 0
       0     .09       0   56.34     .05       0   83.95    .075       0
Bank Sta=56.34,83.95
Exp/Cntr=0.3,0.1

Type RM Length L Ch R = 1 ,70429   ,243.82,256.9,274.66
BEGIN DESCRIPTION:
70351.45
END DESCRIPTION:
XS GIS Cut Line= 6
  909930.6510964   809046.145325  910002.5267166  809063.3330401
  910075.9642047  809069.5825597  910127.5263258  809088.3321426
  910163.4636239  809116.4580533  910221.2762888   809174.269694
#Sta/Elev= 30
       0 1992.97    8.95 1987.19   14.41 1984.55   18.55 1982.72    53.6  1936.5
   61.89 1926.49   64.21 1924.87    71.8 1919.09   73.63  1917.7   84.06 1916.85
   92.15 1916.99  117.03  1917.1  121.22 1917.47  143.92 1920.08  146.43  1920.3
   171.1 1925.54  173.37  1925.7  183.51 1925.89     190 1926.14  201.25 1926.22
  218.96 1927.04   227.7 1927.65  233.13 1928.36  255.74 1930.96  269.41 1934.87
  290.38 1942.21  308.89  1948.1  314.22 1948.75  319.04 1949.13  329.86  1952.7
#Mann= 3 , 0 , 0
       0     .08       0    71.8     .05       0  143.92    .075       0
Bank Sta=71.8,143.92
Exp/Cntr=0.3,0.1

Type RM Length L Ch R = 1 ,70172   ,391.14,376.34,380.67
BEGIN DESCRIPTION:
70094.55
END DESCRIPTION:
XS GIS Cut Line= 6
  909818.1515505  809243.0205545  909894.7137984  809285.2073721
  909941.5892919   809305.519847  909985.3390015  809319.5828023
  910033.7763629  809361.7706441  910057.2135976  809391.4573983
#Sta/Elev= 30
       0 1946.98   10.11 1944.11   13.05 1942.58   27.17  1938.1   50.39 1931.82
   62.08 1929.42   68.53 1927.89   84.33 1925.49   87.64 1925.09   94.25 1923.82
   98.15 1923.46  103.72 1922.28  110.79 1919.51  118.29 1918.41  119.44 1918.37
  131.06 1917.34   138.5 1916.14  156.37 1913.23  160.07 1913.45  162.62 1913.38
  175.43  1913.6  178.46 1913.92  184.46 1916.16  205.12 1923.82  210.87  1925.6
  222.65 1931.22  248.69 1944.49  270.13 1955.85  278.75 1959.88  286.51 1963.36
#Mann= 3 , 0 , 0
       0    .075       0   138.5     .05       0  184.46    .075       0
Bank Sta=138.5,184.46
Exp/Cntr=0.3,0.1

Type RM Length L Ch R = 1 ,69796   ,418.4,414.3,378.44
BEGIN DESCRIPTION:
69718.21
END DESCRIPTION:
XS GIS Cut Line= 4
  909625.9639729  809588.3326278  909758.7759936  809636.7699892
  909819.7134183  809655.5205963  909893.1509064   809750.832427
#Sta/Elev= 30
       0 1944.52    7.87 1940.74   22.93 1937.49   31.06 1935.17   36.38 1934.08
   41.62 1933.32   56.73 1931.43   66.45 1930.52   70.97 1929.76   79.13 1928.91
    84.7 1927.93  102.35  1924.2  106.63 1923.11  110.46 1921.95  140.31 1914.51
  145.35 1914.21  148.13 1913.99  155.86 1913.11   162.2 1911.99  166.13 1911.56
  172.12 1911.75  197.01 1913.16  205.13 1913.96   211.9 1914.41  227.73 1917.35
  255.63 1920.77  257.22 1921.47   292.4 1938.85  307.79    1946  325.45 1951.18
#Mann= 3 , 0 , 0
       0     .07       0  145.35     .05       0   211.9     .08       0
Bank Sta=145.35,211.9
Exp/Cntr=0.3,0.1

Type RM Length L Ch R = 1 ,69382   ,288.24,264.33,244.63
BEGIN DESCRIPTION:
69303.91
END DESCRIPTION:
XS GIS Cut Line= 6
   909568.151308  810010.2079731  909627.5258407  810019.5822525
  909671.2765744  810036.7699676  909691.5890493  810044.5823792
  909743.1511705  810044.5823792  909796.2761837  810071.1453978
#Sta/Elev= 23
       0 1949.51     4.2 1948.01    8.49 1946.35    17.3 1943.47   47.63 1928.23
   52.51 1926.17   58.56  1923.3   90.91 1912.43   99.63 1909.54  104.29 1909.36
  124.91 1909.24  138.68 1909.33  154.88 1912.96  157.77 1913.39  166.53  1914.3
  169.95 1915.02  177.37 1915.78  178.86 1916.02  189.51 1921.22  195.54 1924.66
  208.66 1930.12  225.69 1938.87  239.84 1949.58
#Mann= 3 , 0 , 0
       0     .08       0   90.91     .05       0  154.88    .075       0
Bank Sta=90.91,154.88
Exp/Cntr=0.3,0.1

Type RM Length L Ch R = 1 ,69118   ,194.68,163.8,142.4
BEGIN DESCRIPTION:
69039.58
END DESCRIPTION:
XS GIS Cut Line= 6
  909536.9016617  810308.6455771  909579.0884793  810297.7073816
  909608.7762578  810299.2702735  909646.2764478  810300.8321414
  909691.5890493  810285.2073182  909744.7140625  810249.2700202
#Sta/Elev= 27
       0 1977.33    2.81 1975.65    4.38 1973.99    10.7 1965.24   46.95 1917.39
   48.09 1916.54    52.1 1914.83   57.21 1913.21    67.5 1909.31   74.95 1907.44
   76.29 1906.95   80.89 1907.02   90.83 1906.18   92.95 1906.12   108.5 1907.43
  118.72 1909.86   134.1 1914.42  138.74 1915.49  140.93 1916.21  146.73 1918.53
  158.77 1924.67   165.5 1927.93  190.75  1941.3  195.96 1943.79  212.53 1952.04
  217.82 1956.28  222.91 1959.33
#Mann= 3 , 0 , 0
       0    .075       0    67.5     .05       0  118.72    .085       0
Bank Sta=67.5,118.72
Exp/Cntr=0.3,0.1

Type RM Length L Ch R = 1 ,68954   ,208.25,252.17,262.67
BEGIN DESCRIPTION:
68875.78
END DESCRIPTION:
XS GIS Cut Line= 5
  909635.3392764  810483.6454396  909674.4013342  810463.3329647
  909722.8386956  810430.5204265  909752.5264741  810411.7698194
  909796.2761837  810389.8954767
#Sta/Elev= 26
       0 1946.61    8.33 1939.69   15.16 1933.66    36.6 1917.46   40.28 1913.15
   44.03  1911.7   46.17 1910.86   47.65 1910.61   50.81 1910.27    63.5 1908.11
   67.65  1907.4   75.68 1905.61   80.82 1905.49   82.92 1905.41  102.53  1906.8
  103.19 1906.85  103.26 1906.86  104.691907.459  123.52  1915.3  134.62 1920.16
  137.65 1921.52  139.36 1922.28  171.28 1937.73  176.17 1940.01  182.86 1943.35
  186.56 1944.84
#Mann= 3 , 0 , 0
       0    .075       0    63.5     .05       0  104.69     .09       0
Bank Sta=63.5,104.69
Exp/Cntr=0.3,0.1

Type RM Length L Ch R = 1 ,68702   ,15.94,54.3,80.28
BEGIN DESCRIPTION:
68623.60
END DESCRIPTION:
XS GIS Cut Line= 6
  909705.6509805  810627.3946318  909744.7140625  810658.6453022
  909769.7141892  810664.8948218  909825.9639621  810664.8948218
  909866.5889119  810647.7081308  909925.9634446  810619.5822202
#Sta/Elev= 23
       0  1928.4   27.66 1924.95   31.49 1922.57   50.03 1915.23      65 1909.94
   85.45 1907.18  103.32 1904.72  110.37  1904.2  125.96 1904.11     129 1904.11
  136.84 1904.33  140.47 1904.62  144.39 1906.41  152.41  1909.8  193.49 1933.39
  198.51  1936.7   201.8 1938.75   204.7 1940.76  221.99 1950.17  223.94 1951.33
  224.28 1951.34   236.4 1958.41  241.85 1962.13
#Mann= 3 , 0 , 0
       0    .085       0   85.45     .05       0  144.39    .095       0
Bank Sta=85.45,144.39
Exp/Cntr=0.3,0.1

Type RM Length L Ch R = 1 ,68647   ,33.09,102.96,164.12
BEGIN DESCRIPTION:
68569.30
END DESCRIPTION:
XS GIS Cut Line= 6
  909705.6509805  810639.8946951   909771.276057  810710.2074234
  909804.0885952  810718.0198349  909854.0888486  810721.1456189
  909893.1509064  810732.0827902  909922.8386848  810747.7076134
#Sta/Elev= 26
       0 1926.98    17.7 1924.45    26.7 1923.04   47.88 1912.69    83.4 1909.17
   96.22 1907.79  102.74 1907.37  105.46 1907.32  107.75 1907.12  121.18 1905.14
  126.68 1904.96  142.47 1903.65  150.39 1903.51  154.03 1903.62  160.421905.241
  175.21 1908.99  180.05 1912.27  190.59 1919.61   196.8 1923.16  198.68 1924.32
   206.3 1929.83  217.72 1938.36  220.28 1939.83  232.71  1947.4  241.63 1954.24
  254.16 1963.59
#Mann= 3 , 0 , 0
       0    .085       0  121.18     .05       0  160.42     .09       0
Bank Sta=121.18,160.42
Exp/Cntr=0.3,0.1

Type RM Length L Ch R = 1 ,68544   ,21.93,113.59,138.92
BEGIN DESCRIPTION:
68466.34
END DESCRIPTION:
XS GIS Cut Line= 6
  909697.8385689  810646.1452389  909699.4014609  810691.4578404
  909744.7140625  810744.5828536  909749.4017143  810760.2076767
  909750.9635821  810816.4574496  909757.2141258  810861.7700512
#Sta/Elev= 26
       0 1925.69    3.86 1925.05   45.36 1916.26   47.29 1915.96   53.17 1913.07
   62.49 1912.15  105.28 1907.51  119.54 1905.86  128.76 1903.78  138.79 1903.17
  139.58  1903.2  143.69 1903.01  146.41 1902.71  152.65 1902.21  164.31 1902.12
  167.66 1902.23  173.13 1904.39  180.37  1907.1   187.8 1913.54  200.54 1926.04
  208.66 1930.71  212.04 1933.25  221.35 1939.98  222.77 1940.95  223.74 1941.51
  233.55 1948.87
#Mann= 3 , 0 , 0
       0    .085       0  128.76     .05       0  173.13    .075       0
Bank Sta=128.76,173.13
Exp/Cntr=0.3,0.1

Type RM Length L Ch R = 1 ,68431   ,66.16,58.22,75.96
BEGIN DESCRIPTION:
68352.75
END DESCRIPTION:
XS GIS Cut Line= 6
  909680.6508538  810638.3328273   909677.526094  810668.0206058
   909677.526094  810691.4578404  909668.1518147  810714.8950751
  909632.2134924   810774.270632   909605.651498  810821.1451014
#Sta/Elev= 30
       0 1928.02    5.66 1926.98   21.05 1920.95   29.85 1918.55   49.47 1913.49
   53.29 1912.65   56.69 1911.64   63.62  1910.5   78.53 1908.23   98.29 1905.13
  118.49 1901.93  124.87 1901.78  127.57 1901.68  128.98 1901.63  138.25 1901.46
  146.08 1901.45  147.45 1901.54  147.94 1901.58  154.06 1902.03  154.14 1902.02
  154.35 1902.24  154.66 1902.51  157.18 1904.81  164.81 1911.35  166.58 1914.65
  169.31 1918.17   170.6 1920.72  172.99 1923.82  185.37  1938.1  201.82 1957.61
#Mann= 3 , 0 , 0
       0    .085       0   98.29     .05       0  157.18    .075       0
Bank Sta=98.29,157.18
Exp/Cntr=0.3,0.1

Type RM Length L Ch R = 1 ,68372   ,222.51,279.73,264.83
BEGIN DESCRIPTION:
68294.53
END DESCRIPTION:
XS GIS Cut Line= 6
  909627.5258407  810614.8955926  909613.4639095    810660.20717
  909608.7762578  810711.7703153  909588.4637829  810732.0827902
  909574.4008275  810743.0199616  909543.1511813  810763.3324365
#Sta/Elev= 20
       0 1933.27    6.28 1930.93   47.44 1914.17   52.83 1912.04   87.61    1905
   97.08 1902.88   99.22 1902.61  107.67 1901.24   107.8 1901.23  110.86 1901.08
  119.39 1900.68  123.32 1900.55  127.95  1900.6  128.56 1900.61  130.65 1902.38
     133 1904.37  156.16 1920.73  160.73 1925.63  175.98 1936.63  183.03 1943.32
#Mann= 3 , 0 , 0
       0     .09       0   99.22     .05       0  130.65     .07       0
Bank Sta=99.22,130.65
Exp/Cntr=0.3,0.1

Type RM Length L Ch R = 1 ,68093   ,428.68,420.16,446.53
BEGIN DESCRIPTION:
68014.81
END DESCRIPTION:
XS GIS Cut Line= 6
  909460.3383897   810496.145503  909435.3392872  810527.3951492
  909388.4637936  810546.1447322  909375.9637303  810553.9571437
  909346.2759518  810593.0202257  909330.6511287  810638.3328273
#Sta/Elev= 24
       0  1938.9    13.2 1931.73   22.97 1927.26   38.75 1919.27   40.02 1918.89
   78.79 1905.08    90.5 1901.95   90.71  1901.9   96.531900.292   99.76  1899.4
  104.64 1898.89  104.81 1898.87  105.25 1898.87  112.23 1898.95  117.37 1899.22
  126.19 1899.46  130.87 1900.25   131.2 1900.31   144.4 1903.89  145.26 1903.98
  150.82  1907.2  154.31 1909.08  190.07  1927.8  202.24 1935.29
#Mann= 3 , 0 , 0
       0     .09       0   96.53     .05       0  130.87     .07       0
Bank Sta=96.53,130.87
Exp/Cntr=0.3,0.1

Type RM Length L Ch R = 1 ,67673   ,427.5,419.82,428.58
BEGIN DESCRIPTION:
67594.64
END DESCRIPTION:
XS GIS Cut Line= 6
  909133.7758993  810227.3946533  909086.9014299  810272.7072549
  909015.0258096  810332.0828118  908943.1512136   810419.582231
  908915.0263271  810432.0822943  908852.5260104  810435.2080783
#Sta/Elev= 30
       0 1944.08   14.16 1932.76   26.74  1921.7   41.71  1911.8    61.7 1903.58
   69.98 1903.72   75.47  1902.6   89.06 1903.07  102.71 1902.37  112.17  1901.7
  124.32 1899.82     133 1898.68  142.29 1897.84  156.95 1897.85  164.57 1898.39
  168.87 1898.85  176.76 1900.67  184.35 1901.06  190.93 1902.75  203.95 1902.85
  251.58 1902.33  265.14 1902.51  271.76 1902.41   281.3 1901.71  288.33 1902.09
  313.51 1899.76  317.48 1900.49  328.81 1904.51  340.86 1912.39  365.12 1931.42
#Mann= 3 , 0 , 0
       0    .095       0  124.32     .05       0  176.76    .075       0
Bank Sta=124.32,176.76
Exp/Cntr=0.3,0.1

Type RM Length L Ch R = 1 ,67253   ,298.15,266.6,172.65
BEGIN DESCRIPTION:
67174.83
END DESCRIPTION:
XS GIS Cut Line= 5
  908816.5887124  809949.2705484  908760.3389395  809994.5821258
  908729.0892932  810032.0823158  908683.7766916   810085.207329
  908655.6518052  810125.8322788
#Sta/Elev= 20
       0  1938.8    6.36 1935.22   27.31 1923.79   60.93 1899.15    64.2 1896.72
    66.1 1896.44   80.21 1895.68   91.12 1895.41   99.89 1895.47  106.15 1895.91
  119.65 1898.35  123.41 1898.94  130.14 1899.53  133.19 1899.63   163.3 1899.47
  173.36 1899.16  190.87 1906.95  230.64 1925.32   237.2    1930  240.28 1932.72
#Mann= 3 , 0 , 0
       0    .095       0   60.93     .05       0  119.65    .075       0
Bank Sta=60.93,119.65
Exp/Cntr=0.3,0.1

Type RM Length L Ch R = 1 ,66986   ,122.08,75.95,17.5
BEGIN DESCRIPTION:
66908.23
END DESCRIPTION:
XS GIS Cut Line= 6
  908536.9017155  809811.7698517  908521.2758682  809853.9576935
  908508.7758049  809902.3950549  908505.6510451  809932.0828333
  908513.4634567  810025.8327963  908515.0263487  810094.5826325
#Sta/Elev= 30
       0  1931.8    2.79 1930.23   10.22 1924.98   24.36 1913.01   44.37 1899.45
   57.16 1895.83   68.84 1894.63   79.97 1893.14   82.28  1893.1   87.55 1893.37
   94.92 1893.57   99.36 1893.92  108.21  1895.3  117.83 1896.29  123.82 1897.01
  143.12 1897.88   147.3 1897.51  149.24 1897.47  151.81 1897.26  165.49 1896.91
  177.82 1897.35  200.99 1897.02  210.24 1896.77  213.82 1896.77  223.22 1899.29
  226.03  1899.9  226.82    1900  229.34 1901.86  261.89 1915.03  287.71 1932.86
#Mann= 3 , 0 , 0
       0     .08       0   57.16     .05       0  108.21    .075       0
Bank Sta=57.16,108.21
Exp/Cntr=0.3,0.1

Type RM Length L Ch R = 1 ,66910   ,125.25,112.34,23.37
BEGIN DESCRIPTION:
66832.28
END DESCRIPTION:
XS GIS Cut Line= 6
  908372.8390243  809852.3948015   908433.776449  809896.1455353
  908469.7137471  809928.9580735  908482.2138104  809977.3954349
  908496.2767657  810055.5205747  908504.0891773  810097.7073923
#Sta/Elev= 30
       0 1928.28    7.04 1923.04   11.66 1919.97   18.05 1914.64   45.49 1896.49
   55.251894.681   69.93 1891.96   78.54 1890.93   80.56 1890.94   83.04 1891.43
   89.69 1893.45   93.11  1893.9  104.54 1894.67   114.9 1894.85  128.84 1896.62
  131.72 1897.17   137.6 1897.42   144.1 1897.26  152.58 1896.45  159.98 1896.99
  189.74 1897.31  204.46 1896.45  224.52 1894.87  231.91 1896.95  239.79 1898.11
     260 1914.19  268.82 1917.55  279.52 1924.71  292.19 1929.11  295.99 1931.13
#Mann= 3 , 0 , 0
       0    .075       0   55.25     .05       0  104.54     .07       0
Bank Sta=55.25,104.54
Exp/Cntr=0.3,0.1

Type RM Length L Ch R = 1 ,66798   ,195.03,228.69,210.59
BEGIN DESCRIPTION:
66719.94
END DESCRIPTION:
XS GIS Cut Line= 6
  908305.6510559  809938.3323529  908343.1512459  809983.6449545
  908386.9009555  809999.2697776  908441.5888606  810013.3327329
  908466.5889873  810035.2080998  908486.9014622  810108.6455879
#Sta/Elev= 30
       0 1925.97    3.28 1924.01   24.53 1915.73   31.66 1914.99   36.86 1912.68
   58.82 1901.27   68.52 1896.71   88.62 1895.25   92.06 1894.44  105.27 1892.92
  116.88 1891.63   119.9 1891.16  120.61 1890.82  132.16 1891.34  132.48 1891.46
  149.82 1893.13  161.74 1894.64   167.2 1895.04  171.48 1895.21  175.04 1895.03
  195.53 1895.17  201.67 1895.49  211.56  1898.2  216.01 1899.94  220.14 1903.55
  227.54 1907.73  234.34 1911.86  238.79 1913.95  259.78 1926.85  271.17 1933.36
#Mann= 3 , 0 , 0
       0    .075       0  105.27     .05       0  149.82    .075       0
Bank Sta=105.27,149.82
Exp/Cntr=0.3,0.1

Type RM Length L Ch R = 1 ,66569   ,169.58,188.71,207.65
BEGIN DESCRIPTION:
66491.25
END DESCRIPTION:
XS GIS Cut Line= 5
  908140.0264969   810049.270031  908224.4011563  810135.2075823
  908275.9643016  810180.5201839  908332.2140745  810227.3946533
  908388.4638475  810255.5205639
#Sta/Elev= 30
       0 1933.22    6.88 1929.91   15.93 1924.79   27.83 1918.73   32.56 1916.09
   41.09 1912.56   51.58 1909.71   60.07 1906.35   67.89 1903.71   74.81 1902.08
   83.58 1900.23   94.13  1898.6   99.82 1898.23  116.08 1897.63   124.2  1897.1
  129.19 1897.12  147.52 1896.73  156.65 1896.74  165.71 1897.04  170.76 1896.97
  185.38 1893.39  212.92 1889.91  219.21 1888.74  228.27 1890.95  230.17 1891.86
  258.97 1905.71   293.7 1929.83  305.56 1936.31  320.41 1944.21  325.19 1946.42
#Mann= 3 , 0 , 0
       0     .07       0  185.38     .05       0  230.17     .08       0
Bank Sta=185.38,230.17
Exp/Cntr=0.3,0.1

Type RM Length L Ch R = 1 ,66380   ,332.39,423.79,452.28
BEGIN DESCRIPTION:
66302.53
END DESCRIPTION:
XS GIS Cut Line= 5
  908043.1517741   810160.207709  908086.9014837  810232.0823051
  908140.0264969  810302.3950333  908166.5884913  810335.2075716
  908180.6514467  810382.0830651
#Sta/Elev= 30
       0 1925.39    6.71 1922.59    9.15 1921.48    25.1 1913.82   35.31 1909.47
   39.11 1908.13   52.22 1902.09    56.7 1900.48   67.73 1898.05   70.39  1897.1
   75.88 1895.45    77.5  1895.3   89.99  1894.9  106.72 1894.14  137.53 1893.76
  141.51 1893.65  152.81 1892.99  168.16 1889.93  178.35 1888.42  182.78 1887.99
  194.97 1888.37  212.25 1888.44  214.48 1891.33  214.78 1891.62     246  1942.8
   249.7 1945.75  252.12 1947.88  257.28 1951.42  261.91 1954.86  263.42 1956.26
#Mann= 3 , 0 , 0
       0     .07       0  152.81     .05       0  214.48     .07       0
Bank Sta=152.81,214.48
Exp/Cntr=0.3,0.1

Type RM Length L Ch R = 1 ,65957   ,463.97,440.02,435.11
BEGIN DESCRIPTION:
65878.75
END DESCRIPTION:
XS GIS Cut Line= 5
  907779.0885762  810205.5203106  907761.9008611  810280.5196664
  907738.4636264  810358.6448063  907733.7759746  810405.5202998
  907733.7759746  810461.7700728
#Sta/Elev= 30
       0 1924.84    4.16 1922.85    8.61 1921.17   14.75 1919.39   21.15 1917.33
   38.99 1909.88    48.1 1905.38   51.76 1903.39   68.98 1894.79   79.27 1893.74
   91.27 1891.54  108.63 1891.25   121.1 1890.38   135.9 1889.09   138.1 1888.83
  140.66 1888.11  145.57 1886.97  153.01 1886.01   165.4 1886.04  180.34 1885.92
  187.51 1886.04   197.3 1886.51  205.62 1888.61  216.04 1891.03  224.94 1894.96
  230.51 1898.34  243.92 1906.23  248.36 1908.62  252.97 1910.92  261.87 1916.52
#Mann= 3 , 0 , 0
       0     .08       0  140.66     .05       0  205.62     .07       0
Bank Sta=140.66,205.62
Exp/Cntr=0.3,0.1

Type RM Length L Ch R = 1 ,65517   ,179.14,210.27,249.75
BEGIN DESCRIPTION:
65438.73
END DESCRIPTION:
XS GIS Cut Line= 5
  907310.3387615   810196.145007  907304.0892419  810294.5826218
  907305.6511097  810347.7076349  907305.6511097  810382.0830651
  907294.7139384  810460.2071808
#Sta/Elev= 30
       0 1947.52    5.34  1944.6    8.43 1942.79   17.46 1937.09   19.65 1935.37
   38.49 1921.99   49.17 1911.66   53.73 1909.03   59.01 1908.52   68.06 1896.69
   84.96 1890.13   97.421883.755  100.02 1882.43  107.76  1882.3   127.6 1882.49
  133.761883.785  141.34 1885.45  143.51 1885.79  158.43 1886.95  174.75 1887.59
  185.18 1887.62  194.78 1887.53  209.54 1888.02  222.62 1895.69  231.68 1900.31
  235.42 1902.44  240.64 1906.06  251.18    1914  257.59 1918.55  265.05 1924.37
#Mann= 3 , 0 , 0
       0      .1       0   97.42     .05       0  133.76    .075       0
Bank Sta=97.42,133.76
Exp/Cntr=0.3,0.1

Type RM Length L Ch R = 1 ,65306   ,178.6,195.6,187.44
BEGIN DESCRIPTION:
65228.46
END DESCRIPTION:
XS GIS Cut Line= 6
  907175.9638487  810213.3327222  907132.2141391    810252.39478
   907113.463532  810274.2701469  907085.3386456    810327.39516
  907050.9642395  810371.1448696  907033.7765244  810386.7696927
#Sta/Elev= 26
       0 1922.62    8.03 1919.01   11.39 1918.03    24.2 1909.84   33.03 1905.72
   43.86 1898.78   49.69  1895.6   58.65 1892.43   73.63  1886.9   75.19 1886.69
   77.96 1885.73    79.7  1885.7   89.73 1884.33  106.83 1882.36   117.3 1881.25
   131.1 1881.03  144.64 1881.27  157.92  1881.4  162.32 1883.79  174.86  1890.4
  182.29 1895.44  185.75 1900.17  193.83 1904.78   203.3 1912.37  222.16 1927.28
  226.53 1929.83
#Mann= 3 , 0 , 0
       0     .09       0   89.73     .05       0  162.32    .075       0
Bank Sta=89.73,162.32
Exp/Cntr=0.3,0.1

Type RM Length L Ch R = 1 ,65111   ,365.17,380.63,408.9
BEGIN DESCRIPTION:
65032.85
END DESCRIPTION:
XS GIS Cut Line= 4
  907030.6517646  810099.2702843   906966.588556  810171.1448804
  906935.3389097  810199.2697668  906907.2140232  810264.8948433
#Sta/Elev= 29
       0 1928.17    2.34 1926.67    9.12  1922.3   18.28 1915.69   31.87 1903.13
   35.63 1899.58   42.75 1895.43   51.76 1892.46    67.1 1886.86   73.76 1885.22
   82.29  1884.1    85.7 1883.62   90.32 1882.64   96.28 1881.91  100.59 1881.42
  103.27 1881.01  105.22 1880.87  117.66 1879.88  118.39 1879.88  118.45 1879.87
  130.71 1879.67  131.54 1879.59  138.32 1879.57  149.08 1879.37  151.861881.253
  200.88 1914.45  203.68 1916.42  209.61 1920.92  209.72    1921
#Mann= 3 , 0 , 0
       0      .1       0  105.22     .05       0  151.86    .075       0
Bank Sta=105.22,151.86
Exp/Cntr=0.3,0.1

Type RM Length L Ch R = 1 ,64730   ,470.99,496.19,530.95
BEGIN DESCRIPTION:
64652.22
END DESCRIPTION:
XS GIS Cut Line= 3
    906741.58844  809891.4578835  906649.4013691  809958.6448278
  906561.9009257  810021.1451445
#Sta/Elev= 27
       0 1912.44    2.25 1910.98    8.64 1907.56   37.58 1891.67   38.91 1891.27
   52.21 1886.57   55.46 1885.33   66.51 1884.33   78.29 1882.92   86.55 1881.54
   90.63 1880.94   98.58  1878.4  114.07 1878.14  118.85 1877.59  126.99 1877.14
  130.25 1877.12  141.59 1877.54  142.87 1877.67   153.4 1878.17  159.31 1879.37
  165.11 1882.74  174.89 1889.64  181.97 1892.86   186.2 1895.01  192.94 1897.91
  220.85 1923.88   221.6 1924.48
#Mann= 3 , 0 , 0
       0    .095       0   90.63     .05       0  159.31    .075       0
Bank Sta=90.63,159.31
Exp/Cntr=0.3,0.1

Type RM Length L Ch R = 1 ,64234   ,191.05,216.15,202.6
BEGIN DESCRIPTION:
64156.03
END DESCRIPTION:
XS GIS Cut Line= 4
  906508.7759126  809499.2703166   906410.339322  809536.7705066
  906377.5267838   809546.144786  906304.0892957   809547.707678
#Sta/Elev= 28
       0 1897.78   18.24 1894.31   27.59 1891.97   32.09  1891.1   41.09 1889.69
   48.98 1887.91   63.44 1887.13   64.81 1886.96      78 1884.15   81.33 1883.68
   93.84 1879.27  105.34 1876.33  107.58 1875.77  110.64 1874.79  113.93 1873.87
  121.43 1873.89  133.76 1873.77  136.99 1873.82  139.46 1874.12  154.96 1875.42
   156.31876.155  160.01 1878.19  165.77 1882.48  189.09 1906.26  191.16 1908.17
  191.88 1909.01  211.49 1925.67  212.92 1926.31
#Mann= 3 , 0 , 0
       0    .075       0  105.34     .05       0   156.3    .075       0
Bank Sta=105.34,156.3
Exp/Cntr=0.3,0.1

Type RM Length L Ch R = 1 ,64018   ,143.83,145.11,162.58
BEGIN DESCRIPTION:
63939.88
END DESCRIPTION:
XS GIS Cut Line= 4
  906474.4015065  809325.8323219  906355.6514169  809328.9581058
   906297.838752   809344.582929   906261.901454  809361.7706441
#Sta/Elev= 30
       0 1897.51    1.66 1897.05    9.97 1894.08    29.5 1888.93   34.12 1888.25
   40.72 1886.38    56.2 1882.34   62.75 1881.21   69.28 1880.33   75.02 1879.92
   79.45 1879.51   82.42 1879.34   86.51  1878.9  103.19 1876.66  109.71 1875.69
  113.99 1874.99  118.75 1873.83  120.41 1873.51  122.47 1873.37  139.28 1873.48
  149.18 1875.28  161.53 1876.15  180.19 1885.22  182.82  1886.1   186.3 1888.93
  191.12 1893.18  200.97 1901.46  204.38    1904   212.6 1909.49  218.51 1914.03
#Mann= 3 , 0 , 0
       0    .075       0  109.71     .05       0  149.18    .075       0
#Block Obstruct= 1 ,-1
   25.36    73.91910.102
Bank Sta=109.71,149.18
Exp/Cntr=0.5,0.3

Type RM Length L Ch R = 1 ,63873   ,45.24,54.7,32.02
BEGIN DESCRIPTION:
63794.76
END DESCRIPTION:
XS GIS Cut Line= 5
  906468.1509628   809177.395478  906404.0887783  809188.3326493
  906263.4633218  809188.3326493  906225.9641559  809197.7079529
  906202.5258971  809214.8946438
#Sta/Elev= 30
       0 1910.73    9.63  1906.6   22.87 1901.96   35.65 1895.57   45.15 1890.02
   61.26 1885.12   64.28    1884   71.54  1883.7   83.55 1882.04   97.13 1879.58
   108.5 1875.06  111.86 1874.41  123.39 1873.42  127.78 1872.61  132.12 1872.29
  153.07 1874.22  161.93 1874.89  174.87  1876.7  180.78 1877.58  187.06 1879.07
  202.19 1880.02  204.84 1880.11  207.24 1879.93  216.74 1881.58  222.07 1881.98
  241.91 1890.55  245.74 1892.95  256.82 1899.27  263.44 1904.44  273.33 1910.18
#Mann= 3 , 0 , 0
       0    .075       0  111.86     .05       0  153.07    .075       0
#XS Ineff= 2 , 0
       0   106.5    1882   158.5       0    1882
Permanent Ineff=
       F       F
Bank Sta=111.86,153.07
Exp/Cntr=0.5,0.3

Type RM Length L Ch R = 3 ,63842   ,,,
BEGIN DESCRIPTION:
63765  FBSTR_5034
END DESCRIPTION:
Bridge Culvert--1,0,-1,-1, 0
Deck Dist Width WeirC Skew NumUp NumDn MinLoCord MaxHiCord MaxSubmerge Is_Ogee
22,12,2.6,0, 6, 6, , , 0.95, 0, 1,1,,
       0   116.5   116.5   148.5   148.5     250
    1882    1882    1882    1882    1882    1882
                    1880    1880
       0     132     132     164     164     250
    1882    1882    1882    1882    1882    1882
                    1880    1880
BR Coef=-1 , 0 , 0 ,, 0 ,,,0.8,0,,0,
WSPro=,,,, 1 ,,,, 0 ,,,, 0 ,,,,-1 ,-1 ,-1 , 0 , 0 , 0 , 0 , 0
BC Design=,, 0 ,, 0 ,,,,,,
