HEC-RAS study lds_big_laurel_crk.prj: lds_big_laurel_crk

--- lds_big_laurel_crk.g20 (geometry) --- (continued)

Type RM Length L Ch R = 1 ,63818   ,243.75,140.93,101.58
BEGIN DESCRIPTION:
63740.07
END DESCRIPTION:
XS GIS Cut Line= 6
  906472.8386145  809147.7076995  906407.2135381  809132.0828764
  906340.0265938  809133.6447442  906268.1509735   809139.895288
  906240.0260871  809152.3953513  906191.5887257  809188.3326493
#Sta/Elev= 30
       0 1911.28    6.25  1908.8   13.36 1904.37   19.51 1902.12   28.38 1898.25
   40.67 1889.49   41.96 1888.99   66.77 1883.93   75.21  1882.8   78.32 1882.41
   82.19 1882.53   84.88 1882.14   102.7 1881.47     121 1878.95  133.28 1874.22
  145.37 1872.76  157.29 1872.25   165.7 1872.39  172.93 1873.78  182.34 1874.54
  187.06 1876.98  192.59 1878.11  197.97 1879.69   200.5 1879.83  208.68 1881.25
  217.97 1881.85  239.17 1881.99  258.84 1886.62  267.51 1890.18  297.93 1907.14
#Mann= 3 , 0 , 0
       0    .075       0  133.28     .05       0  172.93    .075       0
#XS Ineff= 2 , 0
       0     117    1881     179       0    1881
Permanent Ineff=
       F       F
#Block Obstruct= 1 ,-1
   49.69   88.591902.933
Bank Sta=133.28,172.93
Exp/Cntr=0.5,0.3

Type RM Length L Ch R = 1 ,63677   ,262.28,256.88,246.31
BEGIN DESCRIPTION:
63599.14
END DESCRIPTION:
XS GIS Cut Line= 6
  906374.4009998  808936.7705389  906327.5265304  808969.5830772
  906272.8386253  809000.8327234  906207.2135488   809044.582433
  906169.7133588   809082.082623  906144.7142563  809133.6447442
#Sta/Elev= 30
       0 1919.47    6.17 1914.75   17.96  1906.6   57.99 1881.17   61.61 1879.49
   66.09 1878.36   81.76 1875.56   89.53 1872.81   94.87 1872.13  115.51 1871.06
  131.03 1872.02  134.73 1872.61  138.36 1873.13  146.04  1873.9  149.46 1874.43
  159.38 1875.39  182.25 1877.17  187.97 1878.33  189.45 1878.47  207.88 1879.49
  215.44  1880.1  219.83 1880.12  227.27 1880.76  233.47  1882.4  241.25 1884.22
  255.31 1887.17  257.56 1887.26  286.11 1900.97  297.79 1906.25  309.45 1910.73
#Mann= 3 , 0 , 0
       0      .1       0   89.53     .05       0  134.73    .075       0
Bank Sta=89.53,134.73
Exp/Cntr=0.3,0.1

Type RM Length L Ch R = 1 ,63420   ,169.46,143.39,117.51
BEGIN DESCRIPTION:
63342.25
END DESCRIPTION:
XS GIS Cut Line= 5
  906196.2763775  808741.4571773  906125.9636492  808791.4574307
   906094.714003  808810.2080377  906072.8386361  808833.6452724
  906047.8385094  808871.1454625
#Sta/Elev= 24
       0 1909.98    6.61 1905.47   13.25 1900.65   21.62 1895.47   48.48 1878.15
   56.68 1872.93   61.57 1871.76   73.16 1870.62   86.95 1869.11  101.81 1869.17
  104.54 1869.34  115.46 1869.75  122.72 1870.87  134.84 1872.47  141.91 1873.52
  148.43 1874.25  154.78 1875.42   155.5 1875.61  175.35 1886.08  176.31 1886.74
  176.92 1886.76  183.27 1887.76  197.61 1893.98  199.85 1895.05
#Mann= 3 , 0 , 0
       0      .1       0   73.16     .05       0  122.72    .075       0
Bank Sta=73.16,122.72
Exp/Cntr=0.3,0.1

Type RM Length L Ch R = 1 ,63277   ,169.01,143.21,67.54
BEGIN DESCRIPTION:
63198.87
END DESCRIPTION:
XS GIS Cut Line= 5
  906060.3385727  808624.2699797  906030.6518185   808675.833125
  905997.8392802  808728.9581381  905969.7133696  808783.6450191
  905952.5266787  808827.3947287
#Sta/Elev= 26
       0 1910.99   51.62 1871.84   64.63 1869.97   72.42 1869.15    75.9 1868.91
   86.18 1868.46   94.43 1868.68  108.06 1869.65  108.89 1869.74  110.73 1870.13
  118.11 1871.43  130.69 1871.87  131.96  1872.1   134.7 1872.37  149.62 1873.49
  153.85 1874.48  156.82 1875.29  163.85 1878.02  175.75 1882.95  183.69  1885.7
  193.63 1888.71  196.68 1889.21  204.74 1890.78  217.44 1895.64  220.81 1896.76
  230.44 1898.45
#Mann= 3 , 0 , 0
       0    .095       0   64.63     .05       0  118.11    .075       0
Bank Sta=64.63,118.11
Exp/Cntr=0.3,0.1

Type RM Length L Ch R = 1 ,63134   ,180.59,144.06,41.65
BEGIN DESCRIPTION:
63055.65
END DESCRIPTION:
XS GIS Cut Line= 4
  905883.7758182  808610.2080485  905879.0891906  808644.5824546
  905879.0891906  808680.5197526  905913.4635967  808813.3327975
#Sta/Elev= 30
       0 1889.98   12.97 1879.16   34.69 1866.59   37.33 1865.07   41.59 1864.95
   43.05 1864.95   51.96 1865.23   62.88 1866.17   66.43 1866.38   66.52 1866.39
   70.63 1866.88   74.75  1867.4   78.33 1867.59   81.48 1868.11    96.5 1870.35
  121.99 1876.05  135.67 1879.04   140.6 1879.77  146.95 1880.78  151.82 1881.67
   153.1    1882  154.08 1882.33  167.16 1885.45  170.77 1885.84  177.74 1888.45
   193.7 1891.54  197.87  1892.3  198.87 1892.73  202.69 1894.03  207.82 1895.98
#Mann= 3 , 0 , 0
       0      .1       0   34.69     .05       0   66.52    .075       0
Bank Sta=34.69,66.52
Exp/Cntr=0.3,0.1

Type RM Length L Ch R = 1 ,62990   ,174.92,161.51,102.5
BEGIN DESCRIPTION:
62911.59
END DESCRIPTION:
XS GIS Cut Line= 5
  905694.7140245  808697.7074677   905760.339101  808718.0199426
  905807.2135704  808741.4571773  905849.4014122  808774.2697155
  905886.9016022  808811.7699056
#Sta/Elev= 30
       0 1943.63    3.93 1937.57    6.09 1935.68   13.63 1928.37   21.12    1917
   36.61 1890.72   37.89 1889.26   39.81 1884.14   45.15  1866.4      48 1865.74
   49.98 1864.24   53.33 1864.46   59.99 1864.16   61.56 1864.29    62.1 1864.19
   71.13 1863.73   86.75 1863.99   108.2 1866.55  114.42 1866.91  122.37 1867.94
  167.56 1876.87  173.01 1877.37   175.1 1877.48  180.26 1878.21  188.35 1879.59
  191.58 1880.52  201.96 1883.87  204.99 1884.69  223.62 1890.89  227.58 1892.11
#Mann= 3 , 0 , 0
       0     .08       0   45.15     .05       0   108.2     .08       0
Bank Sta=45.15,108.2
Exp/Cntr=0.3,0.1

Type RM Length L Ch R = 1 ,62828   ,236.64,244.11,245.37
BEGIN DESCRIPTION:
62750.08
END DESCRIPTION:
XS GIS Cut Line= 5
  905665.0262461  808869.5825705  905719.7141512  808883.6455258
  905741.5884939  808883.6455258  905805.6517026   808878.957874
  905875.9634066  808882.0826338
#Sta/Elev= 25
       0 1910.98   31.55 1878.38      32    1878   41.34 1873.71   45.64 1871.42
    51.9 1869.11   56.47 1867.66   64.47 1865.35   70.96 1864.41   78.34 1863.56
   87.49  1862.5   96.59  1862.2  104.93 1862.25  113.76 1863.54  117.49 1863.92
  121.25 1864.31  128.14 1864.35     134 1864.49  136.71 1864.78  145.94 1867.53
  152.49 1869.28  179.79 1882.92  201.31 1892.56   209.2 1896.46  212.96 1898.49
#Mann= 3 , 0 , 0
       0    .075       0   78.34     .05       0  117.49     .08       0
Bank Sta=78.34,117.49
Exp/Cntr=0.3,0.1

Type RM Length L Ch R = 1 ,62584   ,401.65,424.79,439.93
BEGIN DESCRIPTION:
62505.97
END DESCRIPTION:
XS GIS Cut Line= 6
  905657.2138345  809105.5198577   905721.276019  809121.1446809
  905771.2762723  809124.2704648  905850.9643041  809124.2704648
   905890.026362  809128.9581166  905933.7760716  809166.4572824
#Sta/Elev= 29
       0 1902.56    6.65 1898.53   12.18 1896.37   32.75  1881.7    55.1 1871.94
    59.6 1869.55   65.56 1867.87   71.36  1867.3   76.68 1866.67    84.7 1866.44
   97.89  1866.4  116.04 1862.94  130.93 1860.18  136.77 1860.27  145.18 1860.25
  154.94 1860.07  156.77 1860.17  164.29 1863.68  181.78 1871.68  185.29 1873.06
  208.21 1885.04  225.21  1889.5  231.23  1890.4  240.12 1892.95  250.78 1897.27
  260.68 1899.11  279.68 1907.69  288.37 1910.95  292.69 1912.65
#Mann= 3 , 0 , 0
       0    .075       0  116.04     .05       0  164.29     .08       0
Bank Sta=116.04,164.29
Exp/Cntr=0.3,0.1

Type RM Length L Ch R = 1 ,62159   ,177.34,200.97,204.86
BEGIN DESCRIPTION:
62081.18
END DESCRIPTION:
XS GIS Cut Line= 4
  905574.4010429  809493.0197729  905638.4642516  809516.4580317
  905747.8390376  809552.3953298  905799.4011588   809547.707678
#Sta/Elev= 26
       0 1889.36   10.85  1885.7    23.4 1879.49   34.64 1874.71   43.72 1870.15
   46.08 1869.19   56.75 1865.93    62.3 1864.69   73.49 1863.46   82.47 1863.07
   88.07 1863.07  101.27 1862.79     120 1859.32   122.1 1858.92  127.57 1858.97
  130.47 1858.72  137.78  1858.6  148.94 1858.58  154.35 1858.67   155.91859.658
   174.7 1871.61  183.34 1875.36  189.78 1878.45  201.16 1882.53  221.13 1889.16
  235.12 1897.51
#Mann= 3 , 0 , 0
       0     .07       0     120     .05       0   155.9    .085       0
Bank Sta=120,155.9
Exp/Cntr=0.3,0.1

Type RM Length L Ch R = 1 ,61958   ,31.8,99.74,154.05
BEGIN DESCRIPTION:
61880.21
END DESCRIPTION:
XS GIS Cut Line= 6
  905497.8387951  809608.6451027  905524.4018137  809657.0824641
    905555.65146  809682.0825907  905618.1517767  809719.5827808
  905700.9635441  809749.2705592  905738.4637341  809774.2696617
#Sta/Elev= 30
       0 1891.02   12.23 1888.03   29.18 1884.82   37.88 1882.85   53.71 1878.48
   60.15 1876.42   69.02 1872.22   94.35 1861.12  109.77 1860.02  122.27 1859.37
   126.2 1859.87  128.97 1859.56  139.09 1860.46  152.49 1861.04  160.04 1861.57
     168  1859.1  173.54  1857.2  174.36  1857.1  193.43 1856.18  199.96 1856.25
  206.06 1856.61  219.68 1856.98  227.65 1859.73  239.66 1867.84  259.91 1886.45
  269.96 1894.36  284.67 1903.89  294.64 1910.61  296.85 1911.85  301.19 1915.09
#Mann= 3 , 0 , 0
       0     .07       0     168     .05       0  227.65    .075       0
Bank Sta=168,227.65
Exp/Cntr=0.3,0.1

Type RM Length L Ch R = 1 ,61858   ,26.83,156.52,198.76
BEGIN DESCRIPTION:
61780.47
END DESCRIPTION:
XS GIS Cut Line= 6
  905482.2139719  809614.8956464  905490.0263835  809653.9577043
  905529.0884413   809714.895129  905558.7762198  809743.0200154
  905574.4010429  809763.3324903  905579.0886947  809850.8329337
#Sta/Elev= 30
       0 1889.59   12.66 1886.74   15.47 1885.97   34.83 1881.72   39.35 1880.93
    50.9 1877.71   53.21 1876.74   64.38 1873.11    70.3  1872.8  104.32 1859.46
  117.39 1858.57  123.59 1858.65  150.85 1859.77  157.41 1859.69  161.91 1859.83
  169.21 1859.11  172.37 1858.95  178.74 1858.01  186.79 1857.11  190.79 1856.51
  199.27 1855.35  208.27  1855.5  220.73 1855.49  221.97 1856.46  238.97 1869.75
  244.33 1872.41  249.49 1877.72  261.71 1887.32  264.23 1889.98   266.5 1892.14
#Mann= 3 , 0 , 0
       0    .075       0  190.79     .05       0  221.97    .075       0
Bank Sta=190.79,221.97
Exp/Cntr=0.3,0.1

Type RM Length L Ch R = 1 ,61702   ,425.59,410.51,347.47
BEGIN DESCRIPTION:
61623.95
END DESCRIPTION:
XS GIS Cut Line= 6
  905465.0262568  809613.3327545  905466.5891488  809650.8329445
  905482.2139719  809683.6454827  905393.1516608  809785.2078572
  905380.6515974  809802.3955723  905375.9639457  809827.3946748
#Sta/Elev= 30
       0 1889.99     8.8 1887.12   15.85 1885.19   18.02 1884.33   23.99 1882.39
   26.97 1882.21   28.37 1881.94   37.53 1877.78   45.51 1875.36   55.95 1873.39
   65.35 1871.18   73.88 1868.14   82.41 1864.86   92.27 1859.86   97.06 1858.29
  112.921854.758  116.22 1854.02  127.28 1853.84  129.76 1853.57  141.66 1854.15
  153.88 1854.56  172.41 1855.41  186.95 1857.43  197.82  1860.2  208.27 1867.95
  213.65 1872.21  227.27 1880.24  236.52 1886.24  250.18 1895.57     256 1898.84
#Mann= 3 , 0 , 0
       0    .075       0  112.92     .05       0  153.88    .075       0
Bank Sta=112.92,153.88
Exp/Cntr=0.3,0.1

Type RM Length L Ch R = 1 ,61291   ,73.24,125.64,165.77
BEGIN DESCRIPTION:
61213.44
END DESCRIPTION:
XS GIS Cut Line= 6
  905075.9634497   809622.708058   905054.089107   809658.645356
  905046.2766954  809678.9578309  905044.7138035  809708.6456094
  905044.7138035  809782.0830974  905032.2137401  809822.7080472
#Sta/Elev= 21
       0 1887.65    4.03 1884.66   18.72 1874.56   38.81 1865.51   53.87 1861.14
    62.8 1859.45   76.29 1855.28   83.67 1853.69   94.911850.371   98.64 1849.29
  113.85 1849.24  115.77  1849.3  123.591850.218  143.07  1852.5  157.13    1856
     167 1860.98  173.04 1864.33  177.83 1866.01  188.25 1870.92  196.96 1873.66
  209.51 1877.26
#Mann= 3 , 0 , 0
       0    .085       0   94.91     .05       0  123.59    .075       0
Bank Sta=94.91,123.59
Exp/Cntr=0.3,0.1

Type RM Length L Ch R = 1 ,61166   ,259.71,297.91,321.96
BEGIN DESCRIPTION:
61087.80
END DESCRIPTION:
XS GIS Cut Line= 6
  905024.4013286  809596.1450394  904986.9011385  809630.5204696
  904936.9008852  809683.6454827  904911.9017827  809702.3950656
   904883.775872  809753.9571868  904857.2138776  809766.4572501
#Sta/Elev= 25
       0 1891.94    7.16 1887.46   35.87 1868.49   41.58 1866.24   50.87 1860.39
    52.9 1859.19   87.09 1852.58   93.18 1851.88  104.82 1850.26  123.85 1847.96
   131.3 1846.99  141.85 1847.11  152.34 1847.35  154.46 1847.66  162.01 1848.51
  175.81 1850.28  180.52 1850.76  190.26 1854.02  197.97 1857.32  208.94 1864.16
  220.53 1872.57  222.47 1873.82   229.8 1879.88  233.28 1882.43   243.2 1892.42
#Mann= 3 , 0 , 0
       0     .08       0  123.85     .05       0  162.01    .075       0
Bank Sta=123.85,162.01
Exp/Cntr=0.3,0.1

Type RM Length L Ch R = 1 ,60868   ,440.8,421.56,391.82
BEGIN DESCRIPTION:
60789.89
END DESCRIPTION:
XS GIS Cut Line= 5
  904932.2142576  809383.6449868  904871.2758087  809400.8327019
  904830.6508589  809413.3327652  904802.5259724  809430.5204803
  904750.9638513  809468.0196462
#Sta/Elev= 25
       0 1893.17   27.97  1877.2   32.95 1872.79   51.99 1861.69   60.62 1857.23
   63.32 1856.25    87.1 1847.58   94.76 1844.14   101.4 1843.02   101.7    1843
  103.88 1842.72  105.82 1842.47   110.7 1841.75  111.05 1841.71  118.94 1842.05
  127.98  1842.3  128.45 1842.31  135.63 1842.17  138.78 1842.56  139.47 1842.64
  145.56 1844.65  153.32 1847.81  170.92 1859.52  192.28 1870.92  202.54 1878.79
#Mann= 3 , 0 , 0
       0     .09       0  103.88     .05       0  145.56     .07       0
Bank Sta=103.88,145.56
Exp/Cntr=0.3,0.1

Type RM Length L Ch R = 1 ,60446   ,344.22,250.98,181.32
BEGIN DESCRIPTION:
60368.33
END DESCRIPTION:
XS GIS Cut Line= 6
  904590.0259199  809103.9579899  904525.9637354  809135.2076362
  904500.9636087  809152.3953513  904482.2140258   809174.269694
  904465.0263107  809203.9574725  904446.2767277  809260.2072454
#Sta/Elev= 18
       0 1890.77   10.15 1881.11   56.69 1854.96   58.53 1854.47      76 1841.62
   77.22 1840.91  106.57 1840.71   128.1    1841  139.84 1842.38  142.06 1842.64
  158.58 1846.21  164.73  1847.8  174.13  1850.4  188.55 1861.37  203.71 1871.65
  209.42 1874.66  220.16 1883.05  224.03 1883.96
#Mann= 3 , 0 , 0
       0    .085       0      76     .05       0  139.84     .07       0
Bank Sta=76,139.84
Exp/Cntr=0.3,0.1

Type RM Length L Ch R = 1 ,60195   ,249.96,212.9,125.81
BEGIN DESCRIPTION:
60117.34
END DESCRIPTION:
XS GIS Cut Line= 6
  904229.0890234  809043.0205652  904244.7138465  809097.7074462
  904260.3386697  809153.9572191  904279.0892768   809211.769884
  904279.0892768  809238.3329027  904277.5263848  809283.6455043
#Sta/Elev= 28
       0 1892.13    3.37 1887.83   16.52 1872.68   31.77 1857.63   44.24 1846.66
   51.57 1840.03   56.67 1839.34   56.88 1839.31   63.55  1838.4   71.77 1838.37
   74.49 1838.33   76.15 1838.35   81.36 1838.43      85 1838.52   89.09 1838.55
   97.09 1839.31  108.01 1840.36  115.25 1840.89  139.12 1842.75  166.19 1846.26
  173.42 1847.83  174.27 1848.03  176.03 1848.59  176.89 1848.85   202.6 1859.12
  222.18 1867.01  245.13 1874.29  247.93 1875.47
#Mann= 3 , 0 , 0
       0     .09       0   51.57     .05       0   97.09     .07       0
Bank Sta=51.57,97.09
Exp/Cntr=0.3,0.1

Type RM Length L Ch R = 1 ,59982   ,296.18,307.85,313.51
BEGIN DESCRIPTION:
59904.44
END DESCRIPTION:
XS GIS Cut Line= 6
  904005.6517995  809207.0822322  904063.4634402  809232.0823589
   904107.214174  809258.6453776  904133.7761685  809282.0826123
  904171.2763585  809302.3950872  904232.2137832  809324.2704541
#Sta/Elev= 24
       0 1886.66    6.28 1881.62   13.38 1876.79   28.06 1862.87   30.79 1860.86
   53.18 1839.05   53.52 1838.78   53.83 1838.66   62.99 1837.78   77.31 1836.27
   86.48 1836.61  102.27 1836.52  106.57 1836.57  109.62 1837.67  140.88 1845.44
  152.07 1846.91  169.96  1846.6  174.32  1846.9  184.81 1847.06  206.53 1861.76
  212.12 1865.65  215.44  1867.3  220.68 1869.63  256.99 1882.74
#Mann= 3 , 0 , 0
       0     .08       0   62.99     .05       0  109.62    .075       0
Bank Sta=62.99,109.62
Exp/Cntr=0.3,0.1

Type RM Length L Ch R = 1 ,59675   ,106.18,164.08,203.25
BEGIN DESCRIPTION:
59596.59
END DESCRIPTION:
XS GIS Cut Line= 6
  903877.5264063  809425.8328286  903907.2141848  809480.5197095
   903938.463831  809514.8951397  903985.3393246  809536.7705066
  904004.0889075  809550.8324378  904055.6510287  809605.5203429
#Sta/Elev= 28
       0 1891.01    4.55 1887.66    6.98 1885.38   56.83 1854.69   58.22 1853.67
   62.06 1851.15   75.84 1843.81   78.22  1843.5   81.91 1842.88  108.68 1837.84
  117.28 1836.13  124.35 1835.31  131.03 1834.95  132.35 1834.76  135.11  1834.7
  150.14 1833.84  158.57 1834.03  161.07 1833.92  164.92 1833.99  167.69 1835.33
  180.92 1841.73  189.57  1844.6  208.18 1851.46  215.57 1853.83  235.35 1864.19
   247.8 1870.62   256.2 1875.42  259.01 1877.22
#Mann= 3 , 0 , 0
       0     .08       0  124.35     .05       0  167.69    .075       0
Bank Sta=124.35,167.69
Exp/Cntr=0.3,0.1

Type RM Length L Ch R = 1 ,59510   ,288.5,281.41,273.47
BEGIN DESCRIPTION:
59432.51
END DESCRIPTION:
XS GIS Cut Line= 6
  903794.7136147   809472.707298  903816.5889816  809538.3323744
  903824.4013932  809575.8325645  903822.8385012  809599.2697991
  903836.9014565  809630.5204696  903852.5262796  809678.9578309
#Sta/Elev= 22
       0 1892.77   45.07 1855.37   47.17 1853.39   50.03 1851.15   66.641833.508
   68.06    1832   76.25 1832.07   82.74 1832.39   84.42 1832.29   91.94 1832.16
  123.41 1832.84  130.97 1834.11  153.68 1839.25  155.72 1839.59   163.8 1842.43
  166.84 1843.61  172.82 1847.91  177.26    1851  180.89 1854.45  192.65 1867.73
  207.82 1879.71  216.13 1885.76
#Mann= 3 , 0 , 0
       0     .09       0   66.64     .05       0  130.97    .075       0
Bank Sta=66.64,130.97
Exp/Cntr=0.3,0.1

Type RM Length L Ch R = 1 ,59229   ,232.85,192.82,125.13
BEGIN DESCRIPTION:
59151.10
END DESCRIPTION:
XS GIS Cut Line= 5
  903521.2761374  809466.4577784  903544.7133721  809530.5199629
  903544.7133721  809572.7078047   903568.151631  809653.9577043
  903582.2135621  809702.3950656
#Sta/Elev= 23
       0  1868.2    5.17 1865.58   15.81 1858.61   24.79 1853.57   42.47 1845.01
   48.49 1839.38   53.93 1836.96    70.5 1832.54   79.161830.666   81.08 1830.25
   99.25 1830.43  113.37 1830.42  117.16 1830.35  119.36 1830.44  120.761830.814
   130.1 1833.31  143.26 1836.38  148.54 1837.86  157.82 1841.24  177.95 1848.02
  195.26 1853.72  201.46 1853.59   245.4 1873.29
#Mann= 3 , 0 , 0
       0    .075       0   79.16     .05       0  120.76    .075       0
Bank Sta=79.16,120.76
Exp/Cntr=0.3,0.1

Type RM Length L Ch R = 1 ,59036   ,292.42,270.86,232.51
BEGIN DESCRIPTION:
58958.28
END DESCRIPTION:
XS GIS Cut Line= 4
  903310.3389769  809580.5202162  903346.2762749   809622.708058
   903399.401288  809661.7701158  903500.9636625  809744.5829074
#Sta/Elev= 30
       0 1889.05   18.33 1868.87   20.07 1867.32   29.69 1860.67   43.66 1843.77
   51.43 1833.04   57.33 1829.89   60.99  1829.4   67.75 1828.64   70.72 1828.48
   84.47  1828.3   91.67 1828.34   96.35 1828.55  104.14 1829.23   111.7 1829.87
  123.69 1831.58  126.33 1832.21  137.36 1835.63  147.74 1837.36  164.05 1840.32
  171.79 1841.11  177.28 1841.44   184.3 1842.89  189.89 1844.89  196.02 1846.88
  203.96 1849.01  210.73 1851.05  226.74 1856.74  232.71 1859.36   252.4 1864.56
#Mann= 3 , 0 , 0
       0    .075       0   60.99     .05       0  104.14    .075       0
Bank Sta=60.99,104.14
Exp/Cntr=0.3,0.1

Type RM Length L Ch R = 1 ,58765   ,223.74,241.51,216
BEGIN DESCRIPTION:
58687.42
END DESCRIPTION:
XS GIS Cut Line= 5
  903211.9013621  809875.8330604  903257.2139637  809886.7702317
  903310.3389769  809900.8321629  903374.4011614  809922.7075298
  903408.7765916  809928.9580735
#Sta/Elev= 21
       0 1859.26   10.64 1852.88   14.89 1850.72   18.27 1848.87   31.02 1842.35
   51.43 1830.84   56.64 1829.07   66.59 1827.65   70.47 1827.72   82.09 1827.64
   94.51 1827.36  111.27 1827.26  118.81 1827.07  122.11 1828.42  164.88 1848.36
  169.26 1849.73  180.65 1852.97  184.31 1854.16  191.23 1855.63  203.43 1859.01
   204.2 1859.16
#Mann= 3 , 0 , 0
       0    .075       0   56.64     .05       0  122.11    .075       0
Bank Sta=56.64,122.11
Exp/Cntr=0.3,0.1

Type RM Length L Ch R = 1 ,58524   ,82.94,132.4,191.93
BEGIN DESCRIPTION:
58445.91
END DESCRIPTION:
XS GIS Cut Line= 6
  903105.6513358  810044.5823792  903213.4642541   810121.144627
  903241.5891406  810132.0828226  903310.3389769  810138.3323421
  903382.2135729  810128.9580628  903435.3385861  810111.7703477
#Sta/Elev= 30
       0  1860.5     7.2 1857.22   11.31  1854.6   17.77 1851.23   37.06 1844.64
   44.81 1841.18   45.78 1840.97   67.44 1838.11   95.97 1835.43  116.62 1833.56
  139.91 1832.43  147.28 1831.59   160.5 1829.36  174.35 1826.41   180.9 1825.54
  186.12 1825.02  202.45 1824.65  211.01  1824.7  213.891825.903  222.09 1829.33
  235.89 1832.95  249.09 1837.14  257.03 1837.76  279.61  1837.9  290.21 1838.93
  308.53  1842.6  316.21 1842.98  319.55 1843.53  325.85 1845.86  359.77 1866.83
#Mann= 3 , 0 , 0
       0     .07       0   180.9     .05       0  213.89    .075       0
#Block Obstruct= 1 ,-1
  100.22  138.661847.621
Bank Sta=180.9,213.89
Exp/Cntr=0.3,0.1

Type RM Length L Ch R = 1 ,58391   ,55.83,138.88,184.88
BEGIN DESCRIPTION:
58313.51
END DESCRIPTION:
XS GIS Cut Line= 4
  903057.2139745  810096.1455245   903194.713647  810230.5204373
  903219.7137737  810263.3329755  903252.5263119  810319.5827484
#Sta/Elev= 30
       0 1856.99    5.77 1856.13   10.78 1853.52   14.05 1853.25    19.3 1850.28
   24.57 1848.68   25.79 1848.05   26.78 1846.78   34.12 1838.91   35.53 1838.57
   44.38 1838.24   63.48    1838   69.39 1837.72   77.66  1837.2  106.42 1834.72
  136.61  1831.8  148.19 1830.42  154.07 1830.11  164.31 1829.16  170.98 1827.97
  184.16 1824.97  189.64 1823.81  210.61 1823.71  220.79 1823.47  228.761824.759
  234.18 1825.73  241.66  1831.5  259.21 1849.15  267.52 1855.15  298.63 1872.93
#Mann= 3 , 0 , 0
       0     .07       0  184.16     .05       0  228.76    .075       0
Bank Sta=184.16,228.76
Exp/Cntr=0.3,0.1

Type RM Length L Ch R = 1 ,58253   ,346.95,359.31,326.7
BEGIN DESCRIPTION:
58174.63
END DESCRIPTION:
XS GIS Cut Line= 6
  903022.8385443  810105.5198039  903049.4015629  810157.0829492
  903068.1511458  810189.8954875  903068.1511458  810221.1451337
   903066.589278  810266.4577353  903044.7139111  810335.2075716
#Sta/Elev= 27
       0 1861.74    8.14 1860.25   18.48 1853.88   23.13 1851.18   47.81 1837.75
    66.7 1837.88   73.28  1837.7    74.6 1837.75    82.8 1836.48   90.69 1835.65
   92.58 1835.34    99.7 1833.49  106.49 1831.97  111.59 1830.36  125.56 1826.92
   128.3 1826.08  133.68 1824.03  135.07  1823.5  171.57 1823.46  177.04 1823.23
   179.4 1823.04  182.551823.696  198.04 1827.02  219.61 1839.74   230.3 1847.04
  237.49 1853.14  244.53 1858.77
#Mann= 3 , 0 , 0
       0     .08       0  133.68     .05       0  182.55     .07       0
Bank Sta=133.68,182.55
Exp/Cntr=0.3,0.1

Type RM Length L Ch R = 1 ,57893   ,440.17,424.62,427.86
BEGIN DESCRIPTION:
57815.32
END DESCRIPTION:
XS GIS Cut Line= 6
  902715.0266609  810133.6446904  902705.6513574  810189.8954875
  902708.7761172  810227.3946533  902708.7761172  810275.8330389
  902732.2133519  810350.8323947  902733.7762439  810386.7696927
#Sta/Elev= 29
       0    1869   10.98 1860.19   24.52 1849.74   29.06 1845.23   32.87 1840.86
   56.11 1822.83   61.551821.919   67.06 1820.98   79.98 1820.58    97.2  1820.7
  103.76 1821.39  110.58 1822.36  117.94 1823.41  119.96 1824.08  124.45 1825.36
  133.16 1827.71  143.09 1829.58  149.85 1830.64  165.71 1831.84  176.48 1832.07
  178.48 1832.21  199.81 1834.37  207.98 1835.33  213.53 1836.07  225.64 1838.23
  227.65 1838.75  243.44  1844.6  255.34 1848.31  257.64 1849.34
#Mann= 3 , 0 , 0
       0    .095       0   61.55     .05       0  110.58     .07       0
Bank Sta=61.55,110.58
Exp/Cntr=0.3,0.1

Type RM Length L Ch R = 1 ,57469   ,456.05,418.29,371.89
BEGIN DESCRIPTION:
57390.70
END DESCRIPTION:
XS GIS Cut Line= 6
  902302.5266191  810258.6453237  902310.3390307  810310.2074449
  902310.3390307  810350.8323947  902330.6515056  810411.7698194
  902333.7762654  810483.6454396  902347.8392207  810560.2076875
#Sta/Elev= 28
       0 1855.61   22.68  1844.8    37.2 1837.06   41.23 1834.77   42.37 1834.46
   45.94 1833.75   50.73 1833.08   72.35 1829.78   83.15 1828.45   90.66 1826.41
   92.78 1826.01  102.53 1824.29  121.11  1821.5  123.55 1820.83  135.72 1818.73
  141.04 1818.53  144.74 1818.25  152.32 1818.17  158.86 1818.27  163.971819.962
  178.61 1824.81   199.6 1831.09  205.86    1832  218.45  1834.6  228.98 1836.95
  249.78 1841.22  261.74 1845.78  306.82 1862.15
#Mann= 3 , 0 , 0
       0     .09       0  123.55     .05       0  163.97    .075       0
Bank Sta=123.55,163.97
Exp/Cntr=0.3,0.1

Type RM Length L Ch R = 1 ,57050   ,88.05,143.28,203.44
BEGIN DESCRIPTION:
56972.41
END DESCRIPTION:
XS GIS Cut Line= 5
  901896.2760969  810521.1456297  901938.4639387  810561.7705795
  901952.5258698  810578.9572704  901990.0260599  810638.3328273
   902043.151073    810697.70736
#Sta/Elev= 28
       0 1846.21    7.32  1840.3   24.98 1829.61   42.89 1820.55   51.42 1817.99
   56.37 1815.34   57.21 1815.32   58.57  1815.3   65.08 1815.19   75.37 1815.78
   75.67  1815.8   80.77 1815.89   81.38 1815.89   84.64 1815.94   92.081816.399
   97.45 1816.73  100.06 1816.85  102.33 1817.85  123.01 1826.74  132.02 1830.69
     151 1836.34  159.79 1838.89  167.79 1839.88  194.12 1849.54  211.96  1856.8
  213.25 1857.27  215.89 1858.37  230.67  1863.2
#Mann= 3 , 0 , 0
       0     .09       0   51.42     .05       0  102.33    .075       0
Bank Sta=51.42,102.33
Exp/Cntr=0.3,0.1

Type RM Length L Ch R = 1 ,56907   ,59.29,125.09,193
BEGIN DESCRIPTION:
56829.14
END DESCRIPTION:
XS GIS Cut Line= 5
  901855.6511471  810527.3951492  901835.3386722  810563.3324473
  901821.2767411  810607.0821569  901816.5890893  810638.3328273
  901799.4013742  810727.3951385
#Sta/Elev= 27
       0 1849.75    5.32 1847.45    9.64 1846.04   10.51 1845.54   11.37 1845.26
   34.78 1835.58   57.74 1826.57   72.62 1819.44   75.59 1818.77   82.82  1817.9
   91.281816.046   97.79 1814.64  121.78 1814.71  131.12 1814.66  135.93 1815.42
  137.721815.941  143.52 1817.63   152.4 1820.64  165.95 1823.41  168.22 1824.05
  170.86 1824.91  177.57 1827.68   182.7 1830.04  191.09 1832.76  195.55 1834.85
  208.35 1843.91  209.54 1844.65
#Mann= 3 , 0 , 0
       0    .085       0   91.28     .05       0  137.72    .075       0
Bank Sta=91.28,137.72
Exp/Cntr=0.3,0.1

Type RM Length L Ch R = 1 ,56782   ,163.14,143.92,108.11
BEGIN DESCRIPTION:
56704.04
END DESCRIPTION:
XS GIS Cut Line= 5
  901854.0892793  810499.2702628  901799.4013742  810528.9580412
  901755.6516646  810549.2705161  901704.0885192  810563.3324473
  901665.0264614  810580.5201624
#Sta/Elev= 24
       0 1857.02   10.97 1851.25   34.42 1841.65   38.56 1839.87   62.23 1831.91
   76.13 1827.27   79.84 1826.22   83.13 1824.96  110.46 1816.17  114.91 1814.77
  120.01 1814.28   122.5 1814.37  127.82 1814.55  128.08 1814.55  140.26 1814.42
     143 1814.22  145.66 1814.91  155.091815.458  164.25 1815.99  175.74 1822.25
  190.45 1830.84  197.28 1835.92  205.63 1847.49  206.58 1848.49
#Mann= 3 , 0 , 0
       0     .08       0  110.46     .05       0  155.09    .075       0
Bank Sta=110.46,155.09
Exp/Cntr=0.3,0.1

Type RM Length L Ch R = 1 ,56638   ,260.92,208.34,147.42
BEGIN DESCRIPTION:
56560.12
END DESCRIPTION:
XS GIS Cut Line= 6
   901744.713469  810374.2696294  901694.7142399  810407.0821676
  901668.1512212  810432.0822943  901643.1510945  810463.3329647
  901618.1509679  810508.6455663  901607.2137965  810552.3952759
#Sta/Elev= 28
       0 1847.26   40.46 1821.32   57.351814.167   60.02 1813.04    67.8 1812.85
   69.85 1812.64   86.04  1813.6   89.71 1813.41  101.781814.342  111.48 1815.07
  126.33 1816.45  136.35 1822.41  146.11 1825.65  151.98 1827.25  155.88 1828.41
  158.51 1829.75  160.62 1831.28  167.94 1836.02  171.96 1838.71  175.74 1840.44
  188.25 1848.29  192.24 1850.86  214.29  1862.7  215.99 1862.94  217.59 1863.82
  218.58 1863.99  221.53 1865.98  233.35 1873.34
#Mann= 3 , 0 , 0
       0      .1       0   57.35     .05       0  101.78    .075       0
Bank Sta=57.35,101.78
Exp/Cntr=0.3,0.1

Type RM Length L Ch R = 1 ,56430   ,226.96,265.96,309.62
BEGIN DESCRIPTION:
56351.77
END DESCRIPTION:
XS GIS Cut Line= 6
  901472.8388838  810314.8950967   901469.714124  810378.9572812
  901477.5265355  810418.0203632  901477.5265355  810444.5823577
  901483.7760551  810482.0825477  901491.5884667  810519.5827377
#Sta/Elev= 29
       0 1871.84    6.23 1865.47   10.91 1862.34   54.45  1827.4   54.91 1826.81
   64.13 1815.75   72.16 1814.33   82.16  1812.9   89.74 1812.05   94.33  1811.2
   97.32 1811.05  100.45 1811.16  105.81  1811.1   110.3 1811.16  110.53 1811.16
  116.82 1811.17  128.02 1812.32  130.54  1812.5  136.78 1812.87  148.75 1821.02
  154.88  1825.6  162.68 1829.34   183.5 1840.52  183.77 1840.66  184.98 1841.31
  200.38 1850.25  201.94 1850.93  202.98 1851.41  206.86 1853.92
#Mann= 3 , 0 , 0
       0    .095       0   82.16     .05       0  128.02    .075       0
Bank Sta=82.16,128.02
Exp/Cntr=0.3,0.1

Type RM Length L Ch R = 1 ,56164   ,127.46,176.07,237.29
BEGIN DESCRIPTION:
56085.82
END DESCRIPTION:
XS GIS Cut Line= 5
  901288.4637177  810243.0205006  901246.2758759  810303.9579253
  901222.8386412  810335.2075716  901199.4014065  810372.7077616
    901171.27652  810432.0822943
#Sta/Elev= 26
       0 1863.26   15.59 1850.27    21.5 1844.03   38.09 1831.29   51.67  1820.5
   60.98 1816.81   77.141811.626   80.29 1810.62   85.24 1810.37    91.5 1810.38
  113.18 1810.15  121.161811.122  130.78 1812.33  134.37  1812.9  144.73 1813.74
  155.88 1816.23  161.13  1818.1  170.35 1822.93  173.82 1826.27  184.84 1834.82
  188.98 1838.31  191.26 1840.08  198.39 1844.09   208.1  1851.5  215.21 1857.15
   223.1 1863.97
#Mann= 3 , 0 , 0
       0    .085       0   77.14     .05       0  121.16    .075       0
Bank Sta=77.14,121.16
Exp/Cntr=0.3,0.1

Type RM Length L Ch R = 1 ,55988   ,120.6,240.41,285.94
BEGIN DESCRIPTION:
55909.75
END DESCRIPTION:
XS GIS Cut Line= 6
  901232.2139447  810172.7077724  901143.1516335   810196.145007
  901107.2133113   810216.457482  901080.6513169  810225.8327855
  900997.8385253  810241.4576086  900975.9641826  810260.2071915
#Sta/Elev= 27
       0 1856.31     8.2 1851.71     9.4 1851.13   10.95  1850.1   26.52 1841.14
   31.99 1838.61   38.79 1834.32   53.68 1824.13   61.35 1818.97   63.49 1818.37
   69.02 1818.48   82.27 1817.82  103.18 1816.61   111.5 1814.81   122.3 1813.35
  133.52 1811.26  141.62 1809.84  147.56 1808.53  165.51  1808.3   173.1 1808.52
  177.381811.525  186.63 1818.02  216.09 1840.55  229.49 1849.89  245.96 1853.49
  255.44 1855.82  274.77 1871.24
#Mann= 3 , 0 , 0
       0    .075       0  133.52     .05       0  177.38    .075       0
#Block Obstruct= 1 ,-1
   64.04  111.781831.985
Bank Sta=133.52,177.38
Exp/Cntr=0.3,0.1

Type RM Length L Ch R = 1 ,55747   ,381.97,394.48,384.36
BEGIN DESCRIPTION:
55669.33
END DESCRIPTION:
XS GIS Cut Line= 4
  901229.0891849   810088.333113  901179.0889316  810057.0824425
  901110.3390953  809999.2697776  901069.7141455  809964.8953716
#Sta/Elev= 29
       0 1851.21   26.38 1833.11   43.95 1824.09   46.85 1822.61   54.33 1818.83
   58.96 1816.71   61.04 1815.75   62.99 1815.44   75.87 1813.52    80.8 1812.91
   84.25 1811.87   90.26 1810.52   93.08 1809.61  102.33 1808.27  105.821808.143
  110.03 1807.99  114.27 1808.01  118.35 1808.04  124.39 1807.66  131.77 1807.13
   135.5 1806.67  142.571809.133  146.24 1810.41  148.79 1811.65  166.11 1820.04
  185.93 1838.42  193.74 1847.21  197.88 1854.11  202.01 1858.51
#Mann= 3 , 0 , 0
       0    .075       0  105.82     .05       0  142.57    .095       0
#Block Obstruct= 1 ,-1
   51.89   82.371837.678
Bank Sta=105.82,142.57
Exp/Cntr=0.3,0.1

Type RM Length L Ch R = 1 ,55353   ,437.91,434.4,436.55
BEGIN DESCRIPTION:
55274.85
END DESCRIPTION:
XS GIS Cut Line= 3
  901515.0267255  809857.0824533  901460.3388204  809800.8326804
   901375.964161  809732.0828441
#Sta/Elev= 27
       0 1843.92    6.57 1838.14    11.3 1834.24   21.58 1826.23   29.01 1821.41
   32.26 1818.65   40.84 1813.09   47.83 1810.31   65.11 1805.12   72.21 1803.65
   72.89 1803.51   78.45 1803.72   80.36  1803.8   80.51 1803.81   80.68 1803.81
   85.83 1804.01   91.47 1804.13   101.7 1804.51  119.02 1804.43  124.82  1803.7
  128.38 1803.62  133.55 1805.68  141.25 1808.58  150.27 1813.68  169.61 1827.07
   178.1 1832.06  187.29 1838.81
#Mann= 3 , 0 , 0
       0    .075       0   65.11     .05       0  133.55     .09       0
Bank Sta=65.11,133.55
Exp/Cntr=0.3,0.1

Type RM Length L Ch R = 1 ,54918   ,422.05,421.11,423.43
BEGIN DESCRIPTION:
54840.45
END DESCRIPTION:
XS GIS Cut Line= 3
  901849.4016275  809569.5830449  901732.2134057  809463.3330186
  901688.4636961  809439.8947597
#Sta/Elev= 29
       0 1844.89    5.95 1838.63   14.65 1833.01   14.89 1832.77   14.96 1832.75
   15.29 1832.57   55.91 1807.88   74.13 1805.73    76.5  1805.2   77.39 1805.18
   84.89 1803.97   91.281802.312   95.91 1801.11  107.62 1801.45  108.93 1801.47
   110.7 1801.48  116.83  1801.5  119.51  1801.5  122.79 1801.55  127.17 1801.59
  131.06 1801.56  132.64 1801.63   136.8 1801.91  143.55  1803.4  150.04 1805.01
  151.92 1805.18   155.1 1806.98  158.18 1808.94  207.82 1844.18
#Mann= 3 , 0 , 0
       0    .075       0   91.28     .05       0  143.55     .08       0
Bank Sta=91.28,143.55
Exp/Cntr=0.3,0.1

Type RM Length L Ch R = 1 ,54497   ,371.2,349.95,302.54
BEGIN DESCRIPTION:
54419.33
END DESCRIPTION:
XS GIS Cut Line= 5
  902149.4010993  809272.7073087  902102.5266299  809230.5204911
  902057.2140283  809194.5821689  902022.8385981  809171.1449342
  902000.9642554  809124.2704648
#Sta/Elev= 27
       0 1846.92    7.91 1842.29     9.5 1841.29   23.18  1831.7   38.51 1820.37
   53.91 1806.84    62.8 1801.95   69.871800.598      73    1800    80.3 1798.87
   90.89 1799.17    95.7 1799.57   107.7 1799.72  118.16 1800.16   120.9 1800.49
  126.97 1801.22  131.29 1801.92  141.12 1802.88  143.96 1803.04  157.74 1804.69
  167.04 1806.02  175.87 1811.94  185.21 1820.54   199.3  1832.8   205.7 1840.72
  207.69 1842.64  214.23 1848.55
#Mann= 3 , 0 , 0
       0    .075       0   69.87     .05       0   120.9    .075       0
Bank Sta=69.87,120.9
Exp/Cntr=0.3,0.1

Type RM Length L Ch R = 1 ,54147   ,201.67,159,68.69
BEGIN DESCRIPTION:
54069.39
END DESCRIPTION:
XS GIS Cut Line= 6
  902374.4012152  808950.8324701  902258.7758854  808919.5828238
  902216.5890677  808899.2703489  902194.7137009  808897.7074569
  902158.7764028  808896.1455891  902110.3390415  808903.9580007
#Sta/Elev= 30
       0 1849.62    7.27 1844.01   25.35 1830.61    48.9 1814.13   59.62 1804.48
   68.38 1800.94   74.31 1799.83   80.77 1798.39   82.37 1798.26    86.7 1797.34
   95.28 1797.63  111.64 1797.32  118.08 1797.72  124.16 1797.76  136.19 1799.43
  149.27 1801.06  150.65 1801.06  164.92 1803.18  168.73 1804.02  175.88 1804.82
  180.29 1804.93  185.24 1804.72  190.26 1805.22  197.71 1806.45  202.92 1807.67
  210.76 1812.21  227.56 1820.84  236.32  1827.7  261.26 1842.84  273.56 1851.21
#Mann= 3 , 0 , 0
       0    .075       0   74.31     .05       0  136.19     .07       0
Bank Sta=74.31,136.19
Exp/Cntr=0.3,0.1

Type RM Length L Ch R = 1 ,53988   ,378.8,324.58,205.39
BEGIN DESCRIPTION:
53910.39
END DESCRIPTION:
XS GIS Cut Line= 6
  902335.3391574  808730.5200059  902288.4636638  808763.3325442
  902230.6509989  808799.2698422  902199.4013526  808816.4575573
  902157.2135108  808830.5205127  902108.7761495  808857.0825071
#Sta/Elev= 30
       0 1853.34   17.12 1833.49   29.71 1819.51   38.72 1811.56   46.95  1804.8
   55.741797.944   57.86  1796.3   69.97 1796.07   82.55 1796.31   87.19 1796.57
   95.81 1797.36   98.99 1797.64  110.39 1799.39   122.4  1800.1  131.23  1800.4
  133.25  1800.6  137.73 1801.47  151.65 1803.29  157.89 1804.58   166.5 1805.36
  175.27 1806.73  177.63 1807.39  182.97 1808.34  191.98 1811.63  201.71 1815.48
  209.54 1819.49  212.67 1821.44  234.59 1833.02  253.74 1842.69  260.67  1846.8
#Mann= 3 , 0 , 0
       0      .1       0   55.74     .05       0   95.81    .075       0
Bank Sta=55.74,95.81
Exp/Cntr=0.3,0.1

Type RM Length L Ch R = 1 ,53664   ,317.42,265.14,125.95
BEGIN DESCRIPTION:
53585.81
END DESCRIPTION:
XS GIS Cut Line= 6
  901994.7137116  808525.8323649  902004.0890152  808574.2697263
  902004.0890152  808625.8328716  902002.5261232  808664.8949295
  902000.9642554   808710.207531  901997.8384714  808797.7079744
#Sta/Elev= 30
       0 1833.18    4.96 1827.75   25.22 1816.01   36.04 1806.77    38.9 1803.42
   47.82  1797.4    56.71796.062   64.18 1794.97   66.93 1793.92   81.31 1793.72
   94.59 1794.32   99.34 1794.94  103.721795.765  110.18 1796.99  118.59 1797.67
  124.66 1799.18  128.28  1799.6  138.58 1801.37     149 1801.94  152.16  1802.5
  159.06 1804.44   167.6 1806.14  196.83 1807.27  207.32 1811.11  225.38 1819.03
  231.31  1822.1  244.88 1829.95  256.99 1835.32  265.34 1838.12  272.89 1842.61
#Mann= 3 , 0 , 0
       0    .085       0    56.7     .05       0  103.72     .07       0
Bank Sta=56.7,103.72
Exp/Cntr=0.3,0.1

Type RM Length L Ch R = 1 ,53399   ,386.85,391.64,389.38
BEGIN DESCRIPTION:
53320.67
END DESCRIPTION:
XS GIS Cut Line= 6
  901683.7760443  808596.1450932  901727.5267781  808614.8946761
  901808.7766777  808666.4578215  901849.4016275   808710.207531
  901879.0883818  808752.3953728  901893.1513371   808803.957494
#Sta/Elev= 30
       0 1865.99   26.81  1841.8   42.66  1814.7    47.6 1807.49    55.4 1796.64
   58.241794.724    60.5  1793.2   65.82 1792.99   69.29 1792.42   82.73 1792.51
   89.78 1792.84  100.651794.275  120.75 1796.96  128.73 1798.21  130.16 1798.29
  139.53 1797.82  147.17 1797.91  150.53 1797.65  157.62 1798.13  175.97 1800.37
  200.24 1802.06  211.73 1803.07   226.2 1808.07  235.48 1811.05  251.67 1818.89
  255.12 1820.64  271.77 1830.33  279.18 1835.63   297.9 1846.26  308.57 1851.53
#Mann= 3 , 0 , 0
       0    .075       0   58.24     .05       0  100.65     .07       0
Bank Sta=58.24,100.65
Exp/Cntr=0.3,0.1

Type RM Length L Ch R = 1 ,53007   ,275.13,283.6,282.88
BEGIN DESCRIPTION:
52929.03
END DESCRIPTION:
XS GIS Cut Line= 6
  901449.4016491  808872.7073303  901511.9009416  808919.5828238
  901536.9010683  808938.3324067  901575.9641502  808977.3954887
  901607.2137965  809014.8946546  901643.1510945   809044.582433
#Sta/Elev= 30
       0 1842.37    5.14 1839.03   22.66 1823.01   25.08 1821.79   29.46 1819.22
   55.35 1806.16   67.77 1802.73   90.57 1795.01   95.01 1794.37   99.09 1794.45
  107.18  1793.8  115.24 1792.41  118.26 1791.86  122.97 1791.36  126.21 1791.16
  137.15 1790.75  143.66 1790.83  149.56 1791.06  153.22 1790.93  157.511792.428
  164.62 1794.97  168.58  1796.5  195.98 1813.05  207.31 1818.95   220.5    1830
  229.59 1841.48  236.62 1849.77  241.23 1852.47  242.96 1854.05  260.05 1866.95
#Mann= 3 , 0 , 0
       0    .075       0  115.24     .05       0  157.51    .075       0
Bank Sta=115.24,157.51
Exp/Cntr=0.3,0.1

Type RM Length L Ch R = 1 ,52723   ,75.57,92.1,123.03
BEGIN DESCRIPTION:
52645.42
END DESCRIPTION:
XS GIS Cut Line= 6
  901268.1512427  809041.4576732   901300.963781  809099.2703382
  901325.9639077  809125.8323326  901357.2135539  809160.2077629
  901382.2136806  809182.0831297  901416.5891108  809232.0823589
#Sta/Elev= 28
       0 1832.46    3.04 1830.45   12.49 1825.15   21.44 1820.87   41.83 1809.76
   58.61 1801.23   68.86 1797.39   71.46 1796.15   82.59 1794.06   96.55 1790.74
  102.95 1789.87  114.75 1788.29  126.31 1788.48  137.51 1788.77  143.38 1789.23
  147.91  1790.1  149.41 1790.65  159.06 1794.29   170.3  1796.8  182.93 1803.26
  198.73 1813.12  201.33 1814.63  206.02 1817.58  218.35 1826.29  219.62  1827.3
  223.58 1830.22  240.34 1841.37   243.3 1843.75
#Mann= 3 , 0 , 0
       0    .075       0  102.95     .05       0  149.41    .075       0
Bank Sta=102.95,149.41
Exp/Cntr=0.3,0.1

Type RM Length L Ch R = 1 ,52631   ,76.93,90.87,102.51
BEGIN DESCRIPTION:
52553.32
END DESCRIPTION:
XS GIS Cut Line= 6
  901213.4633376  809072.7073195  901232.2139447  809122.7075728
  901268.1512427  809191.4574091  901274.4017865  809214.8946438
  901279.0884141  809243.0205545  901290.0266096  809294.5826756
#Sta/Elev= 29
       0 1827.61    1.02 1826.97    1.49 1826.78   10.06 1823.72   11.74 1822.87
   16.23 1819.67   34.93 1808.88   46.78 1802.42    53.4 1800.72   80.92 1793.89
   88.34 1792.22   97.67 1790.17  104.35 1789.98  107.39 1789.94   114.9 1789.66
  122.781788.558  130.96 1787.42  148.34 1786.49  155.24 1788.32  162.22 1790.27
  163.64 1790.43  166.41 1792.58  180.93 1806.44  183.76 1808.77  196.27 1819.15
   203.3 1823.51  221.35 1838.73  235.46 1851.68  236.47 1852.48
#Mann= 3 , 0 , 0
       0    .075       0  122.78     .05       0  155.24     .07       0
Bank Sta=122.78,155.24
Exp/Cntr=0.3,0.1

Type RM Length L Ch R = 1 ,52540   ,290.86,303.51,280.58
BEGIN DESCRIPTION:
52462.45
END DESCRIPTION:
XS GIS Cut Line= 6
  901158.7764567  809093.0197944  901163.4641084  809150.8324593
  901179.0889316  809186.7697573  901182.2136914  809216.4575358
  901180.6518236  809274.2702007  901194.7137547  809307.0827389
#Sta/Elev= 26
       0  1831.2     .69 1830.98    2.78    1830      46 1811.26      58 1806.53
   62.51 1804.95    66.6 1804.42    73.6 1801.87   88.84 1793.21   97.19 1790.77
   99.75 1789.93  104.14 1789.66  109.58 1788.98  121.67 1787.18  129.13  1785.9
  131.24 1786.25  142.99 1786.98   143.7 1786.97  148.92  1788.9  160.47 1793.29
  170.85 1799.97  191.31 1813.32  192.96 1814.28  195.04 1815.62  204.61 1823.83
  220.61 1838.04
#Mann= 3 , 0 , 0
       0    .075       0  109.58     .05       0  148.92     .07       0
Bank Sta=109.58,148.92
Exp/Cntr=0.3,0.1

Type RM Length L Ch R = 1 ,52237   ,384.39,393.56,411.09
BEGIN DESCRIPTION:
52158.95
END DESCRIPTION:
XS GIS Cut Line= 6
  900877.5265678  809125.8323326  900877.5265678  809202.3956046
  900882.2142196  809236.7700107   900891.588499  809264.8948972
  900900.9638025  809289.8950238  900902.5266945  809330.5199736
#Sta/Elev= 22
       0 1830.56    2.89  1829.5   30.07 1808.84   34.45 1803.21   38.92 1800.02
    62.61787.114   64.46  1786.1   64.85 1785.81   65.47 1785.75   76.56 1785.78
   81.33 1785.63   91.25 1785.74   98.73 1786.72  117.29 1788.96  121.79 1789.31
   140.9 1791.34  149.02 1791.18  153.72 1791.21  166.05 1795.13  177.08 1801.06
  183.73 1805.31  208.26 1822.74
#Mann= 3 , 0 , 0
       0    .095       0    62.6     .05       0   98.73     .07       0
Bank Sta=62.6,98.73
Exp/Cntr=0.3,0.1

Type RM Length L Ch R = 1 ,51843   ,364.52,359.98,339.01
BEGIN DESCRIPTION:
51765.39
END DESCRIPTION:
XS GIS Cut Line= 6
  900504.0885839   809138.332396  900490.0266527  809196.1450609
  900490.0266527  809219.5822956  900490.0266527  809253.9577258
  900490.0266527  809299.2703274  900496.2761723  809346.1447968
#Sta/Elev= 29
       0 1817.14   17.63 1806.06   22.89 1803.01   31.09 1798.54   40.41 1795.14
   44.33 1793.87   48.06 1792.82   51.74  1791.9   55.58 1791.26   65.33 1789.86
   68.11 1789.72   82.94 1787.54  102.11 1784.72  105.59 1784.03  116.39 1784.07
  133.45  1784.3  138.35 1784.49  141.761786.415     153 1792.76  156.03 1793.75
     173 1805.98  178.51 1810.48   179.9 1811.43  181.31 1812.28  189.59 1816.94
  197.41 1822.82  202.09  1826.5  208.41 1830.72  209.91 1831.85
#Mann= 3 , 0 , 0
       0     .09       0   82.94     .05       0  141.76     .07       0
Bank Sta=82.94,141.76
Exp/Cntr=0.3,0.1

Type RM Length L Ch R = 1 ,51483   ,208.98,171.98,114.77
BEGIN DESCRIPTION:
51405.41
END DESCRIPTION:
XS GIS Cut Line= 6
  900136.9011436  809146.1448075  900132.2134919  809183.6449976
   900130.651624  809221.1451876   900130.651624  809252.3948338
  900135.3392758  809308.6456309   900186.901397  809388.3326386
#Sta/Elev= 29
       0 1831.64   11.23  1822.9   19.47 1813.41   27.71 1805.63   38.17 1797.38
   64.69  1787.4   87.47 1781.78   98.71 1782.51  105.46 1783.94  112.53 1785.23
  120.76 1787.04  133.36 1787.32  139.82 1787.54   146.8 1788.02   149.5 1788.35
   158.5 1789.85  172.74 1792.78  181.15 1794.45  183.77  1794.9  197.38 1798.19
  207.46 1800.43  213.19 1801.27  220.76 1803.11  227.35 1804.86  234.73  1806.6
  239.46 1807.47  242.55 1808.35   256.9 1813.07  257.95 1813.33
#Mann= 3 , 0 , 0
       0    .095       0   64.69     .05       0  120.76    .075       0
Bank Sta=64.69,120.76
Exp/Cntr=0.3,0.1

Type RM Length L Ch R = 1 ,51311   ,252.1,227.48,148.7
BEGIN DESCRIPTION:
51233.43
END DESCRIPTION:
XS GIS Cut Line= 6
  899911.9010277  809185.2078895  899930.6516348  809225.8328393
  899957.2136293  809258.6453776  899997.8385791  809313.3322585
  900030.6511173  809360.2077521  900100.9638456  809461.7701266
#Sta/Elev= 30
       0 1862.14     7.3 1857.15    18.7 1843.95   44.74 1807.35   48.39 1802.35
   60.44 1788.69   65.47 1783.35   74.76 1781.21   88.07  1780.3  108.25 1780.55
  109.91 1780.68  112.56 1780.59  114.07 1781.17  119.311782.573  127.93 1784.88
  138.81 1785.35  150.17 1786.41  154.85  1786.7  170.77 1788.81  179.98 1790.56
  188.91 1791.55  194.06 1791.82   205.6 1792.83  221.81 1793.58  231.71 1793.87
   255.4 1795.65  287.39 1800.48  315.52  1815.8  325.95 1820.43  335.83 1825.79
#Mann= 3 , 0 , 0
       0     .09       0   65.47     .05       0  119.31    .075       0
Bank Sta=65.47,119.31
Exp/Cntr=0.3,0.1

Type RM Length L Ch R = 1 ,51084   ,358.01,408.04,455.33
BEGIN DESCRIPTION:
51005.95
END DESCRIPTION:
XS GIS Cut Line= 5
  899732.2135134  809399.2698099  899791.5890703  809432.0823482
  899930.6516348  809485.2073613  899969.7136926   809510.207488
  899997.8385791  809541.4571342
#Sta/Elev= 30
       0    1835   10.55 1827.84   21.08 1817.74   31.37 1810.24   36.22 1807.39
   45.42 1801.13   51.22  1796.3   62.48 1790.28    69.7 1786.07   74.45 1783.79
   78.02 1782.99   82.44 1781.98  111.81 1780.16  123.49  1780.5  132.77 1781.25
  137.961781.927  144.54 1782.82   157.1 1785.81  167.94 1786.73  174.76 1787.82
  182.23  1788.6  199.98 1791.71  212.79 1793.52  227.83 1796.15  249.41 1802.84
  254.24 1802.44  259.04 1804.03  263.08 1806.05  282.45 1816.92  305.12 1827.47
#Mann= 3 , 0 , 0
       0     .08       0   78.02     .05       0  137.96    .075       0
#Block Obstruct= 1 ,-1
  155.04  173.37 1797.59
Bank Sta=78.02,137.96
Exp/Cntr=0.3,0.1

Type RM Length L Ch R = 1 ,50676   ,454.84,454.02,462.41
BEGIN DESCRIPTION:
50597.91
END DESCRIPTION:
XS GIS Cut Line= 5
  899500.9638779  809618.0204062  899524.4011126  809680.5196988
  899552.5259991  809724.2704325  899571.2766062  809753.9571868
  899621.2758353  809822.7080472
#Sta/Elev= 26
       0 1815.27    4.05 1812.68    8.55 1810.03    20.2 1802.18   35.15  1794.5
   45.61 1790.79   52.29  1787.9    58.6 1786.81   64.78 1785.18   71.58 1783.78
   76.76 1782.77   78.11 1782.57   82.02 1781.19   83.41 1780.91   87.21 1780.47
  114.21 1778.74  118.68 1778.63  124.79  1778.7  125.98 1778.65  130.88 1781.33
  167.29 1801.26  184.78    1810  188.58 1812.14  191.06 1813.75  237.68 1840.15
  238.88 1841.02
#Mann= 3 , 0 , 0
       0     .08       0   87.21     .05       0  130.88    .075       0
Bank Sta=87.21,130.88
Exp/Cntr=0.3,0.1

Type RM Length L Ch R = 1 ,50222   ,179.04,244.59,276.55
BEGIN DESCRIPTION:
50143.89
END DESCRIPTION:
XS GIS Cut Line= 5
  899113.4639628  809849.2700417  899135.3383055  809897.7074031
  899149.4012608  809936.7704851  899177.5261473  809972.7077831
  899188.4633186  810053.9576827
#Sta/Elev= 26
       0 1826.76   11.22 1818.48   23.23 1807.92   36.21 1796.17   53.15 1784.01
    55.2 1782.51    58.8 1781.77   65.21 1780.92   79.221777.882   82.391777.195
   85.32 1776.56   93.94 1776.53    94.8 1776.53  102.58  1776.6  103.71 1776.62
  108.29 1776.57  112.81 1776.54  120.52 1776.54  126.48 1776.51  131.261777.419
  134.53 1778.04   140.3 1781.12  148.08 1785.79  162.43  1795.1  169.97 1796.64
  222.28 1822.25
#Mann= 3 , 0 , 0
       0     .08       0   82.39     .05       0  131.26    .075       0
Bank Sta=82.39,131.26
Exp/Cntr=0.3,0.1

Type RM Length L Ch R = 1 ,49977   ,188.75,184.76,196.83
BEGIN DESCRIPTION:
49899.30
END DESCRIPTION:
XS GIS Cut Line= 6
  899004.0891767  809869.5825166  898957.2136831  809916.4580102
    898941.58886  809936.7704851  898927.5259047  809961.7706118
  898927.5259047  809980.5201947  898908.7763218  810102.3950441
#Sta/Elev= 30
       0 1807.97    5.72 1805.72   22.13 1802.07   27.04 1799.95   48.52 1794.68
   54.31  1793.9   59.68 1791.75   64.99 1788.96   77.24 1781.56   91.17 1780.23
  103.06 1778.12  117.38 1777.15   120.6 1776.81  134.36 1776.22  139.35 1775.48
  143.84 1774.79  158.99 1774.38  172.93 1774.53  185.46 1774.89  188.531776.983
  189.86 1777.89  192.61 1781.06  214.54  1800.1  220.34  1804.9  224.65 1808.27
  229.64 1811.25  235.79 1816.13  242.01 1821.17  244.94 1823.37  262.67  1836.1
#Mann= 3 , 0 , 0
       0    .075       0  139.35    .045       0  188.53     .07       0
Bank Sta=139.35,188.53
Exp/Cntr=0.3,0.1

Type RM Length L Ch R = 1 ,49792   ,429.3,414.46,395.08
BEGIN DESCRIPTION:
49714.54
END DESCRIPTION:
XS GIS Cut Line= 5
  898794.7138839  809833.6452186  898758.7765859  809925.8322896
  898740.0259788  809977.3954349  898722.8392879  810007.0821892
  898710.3392245  810046.1452712
#Sta/Elev= 27
       0  1802.7    4.56 1800.78    7.72 1799.19   38.18 1785.46   47.38 1781.89
   52.82 1780.59   58.97 1780.17   73.31 1779.02   75.88 1778.92   86.43 1777.99
   95.24 1776.31  101.76 1774.28  110.56 1774.23  114.83 1774.13   119.6 1774.22
   131.7 1774.09  142.96 1774.17   145.41775.969   156.1 1783.84  185.86 1801.87
  188.57 1802.42  193.24 1805.59  201.77 1808.78  202.55 1809.36  211.87  1817.5
  216.53 1824.21  229.13 1838.37
#Mann= 3 , 0 , 0
       0     .08       0   95.24    .045       0   145.4     .07       0
Bank Sta=95.24,145.4
Exp/Cntr=0.3,0.1
