HEC-RAS study lds_big_laurel_crk.prj: lds_big_laurel_crk

--- lds_big_laurel_crk.g20 (geometry) --- (continued)

Type RM Length L Ch R = 1 ,49378   ,362.58,315.11,202.04
BEGIN DESCRIPTION:
49300.08
END DESCRIPTION:
XS GIS Cut Line= 5
  898375.9643225  809724.2704325   898365.026127  809816.4575035
  898350.9641959  809886.7702317  898346.2765441  809933.6447011
  898346.2765441  809977.3954349
#Sta/Elev= 25
       0 1826.25   26.48  1799.3   52.55  1775.3   65.68  1771.5    70.2  1771.7
   76.28 1771.82   83.55 1771.84   84.72 1771.93   98.26 1773.34  107.91 1774.88
  113.98 1775.63  123.29 1777.12  126.26 1777.66  133.07 1779.09  140.32 1780.31
  146.85 1781.02  154.17 1782.04  177.46 1784.28  192.11 1785.95  195.52 1786.19
  202.66 1786.97  211.79 1788.32  226.29 1794.86  254.58 1802.95   255.4 1803.25
#Mann= 3 , 0 , 0
       0      .1       0   52.55     .05       0  107.91     .08       0
Bank Sta=52.55,107.91
Exp/Cntr=0.3,0.1

Type RM Length L Ch R = 1 ,49063   ,440.92,502.1,542.83
BEGIN DESCRIPTION:
48984.97
END DESCRIPTION:
XS GIS Cut Line= 6
   897996.276819  809746.1447752  898050.9636999  809803.9574402
  898090.0267819  809874.2701684  898144.7136629  809950.8324162
  898158.7766182  809978.9573027  898166.5890298  810039.8947274
#Sta/Elev= 30
       0 1841.06   17.16 1825.93   29.27 1816.66   45.63 1797.79   48.46 1793.29
   59.71 1774.17   61.53 1773.36   74.23 1770.46   82.19 1770.07   88.36 1769.97
   98.05 1770.04  119.95  1773.2  130.17 1774.53  139.56 1776.03  146.97 1776.69
  175.48 1777.94  188.55 1778.32  201.54  1779.4  212.59 1780.85  228.51 1782.57
  236.89  1783.3     258 1786.14  264.52 1787.18  271.49 1789.23  273.72 1790.12
  285.65 1793.36  299.64 1797.57  317.73 1803.99  337.57 1809.84  347.09 1813.76
#Mann= 3 , 0 , 0
       0     .08       0   59.71     .05       0  119.95     .07       0
Bank Sta=59.71,119.95
Exp/Cntr=0.3,0.1

Type RM Length L Ch R = 1 ,48561   ,77.26,138.4,172.13
BEGIN DESCRIPTION:
48482.87
END DESCRIPTION:
XS GIS Cut Line= 6
  897665.0266768  809872.7072764  897616.5893154  809950.8324162
  897608.7758797   809993.020258  897605.6511199  810025.8327963
  897652.5266134  810127.3951708  897633.7760064   810197.707899
#Sta/Elev= 30
       0 1809.05    2.75 1806.82   23.02 1794.73   35.06 1788.87   38.61 1787.36
   51.69 1780.44   66.68 1778.65   91.98 1778.04  114.72 1777.04  125.22 1776.42
  162.09 1775.14  169.63 1773.31  179.18 1771.76  182.12 1771.04  186.16 1770.57
  190.631769.731  199.21 1768.12  205.66 1767.81  217.22 1767.82  231.58 1768.07
  240.01 1768.76   259.2 1771.74  271.75 1772.95  283.31 1773.31  301.95 1785.53
  316.72 1795.75  318.12 1796.35  321.67 1798.75   328.8 1801.91     354 1814.12
#Mann= 3 , 0 , 0
       0    .085       0  190.63     .05       0   259.2     .06       0
Bank Sta=190.63,259.2
Exp/Cntr=0.3,0.1

Type RM Length L Ch R = 1 ,48422   ,234.9,306.82,324.25
BEGIN DESCRIPTION:
48344.46
END DESCRIPTION:
XS GIS Cut Line= 6
  897594.7139485  809849.2700417  897540.0260434  809946.1447645
  897513.4640489  810011.7698409  897499.4010936  810053.9576827
  897486.9010303  810138.3323421  897465.0266876  810185.2078357
#Sta/Elev= 30
       0 1808.49   20.88 1793.87   27.53 1789.55   37.57 1784.58   48.81 1779.75
   51.72 1779.13   81.09 1777.56   90.37 1777.78  110.56 1777.34  127.33 1777.25
   141.6 1776.95  156.14 1777.01  167.38 1776.25  185.03 1775.65  207.43 1773.53
  214.73 1772.19  219.43 1771.64  236.02 1771.34  241.33 1771.13  254.57 1769.54
  258.56 1768.88  267.37 1767.55  280.97 1767.15  294.97 1767.05   304.1 1768.74
  318.41 1783.73  320.41 1786.24  334.95 1799.23  349.11 1812.38  364.14 1825.84
#Mann= 3 , 0 , 0
       0     .07       0  258.56     .05       0   304.1     .06       0
#Block Obstruct= 1 ,-1
   181.6  221.741789.856
Bank Sta=258.56,304.1
Exp/Cntr=0.3,0.1

Type RM Length L Ch R = 1 ,48116   ,291.19,178.71,117.49
BEGIN DESCRIPTION:
48037.65
END DESCRIPTION:
XS GIS Cut Line= 6
  897377.5262442  809777.3954457  897352.5261175   809825.832807
  897240.0265716  809941.4581369  897193.1510781  810002.3955616
   897177.526255  810032.0823158  897169.7138434  810057.0824425
#Sta/Elev= 30
       0 1805.91    3.67 1803.45   16.89 1796.03   20.44 1793.79    31.9 1785.76
   37.28  1782.5   44.11  1779.4   49.49 1778.03    65.1 1776.97   78.04 1776.34
  105.87 1775.81  133.09 1774.36   160.6 1772.32  187.31 1770.88  200.74 1769.85
  208.03 1768.16  214.66 1766.58  216.09 1766.52  228.65 1766.29  256.86 1766.23
  265.03 1766.36  266.881767.818  280.71 1778.72  292.26 1786.48  301.58 1792.12
  310.02  1796.3  327.13 1803.51  334.95 1806.58  337.29 1807.94  352.65 1815.56
#Mann= 3 , 0 , 0
       0     .07       0  208.03     .05       0  266.88    .065       0
Bank Sta=208.03,266.88
Exp/Cntr=0.3,0.1

Type RM Length L Ch R = 1 ,47937   ,200.62,130.92,22.68
BEGIN DESCRIPTION:
47858.94
END DESCRIPTION:
XS GIS Cut Line= 6
  897041.5884502  809774.2696617  897065.0267091  809843.0205221
  897069.7133367  809872.7072764  897069.7133367  809941.4581369
  897075.9638804  809978.9573027  897097.8392473  810058.6453345
#Sta/Elev= 30
       0 1801.54   13.09 1794.92   27.97 1788.58   42.39 1784.16   48.25 1782.23
   55.53  1779.2   80.451766.269    84.9    1764   88.12 1763.87  105.69 1764.22
  120.04    1765  126.36 1765.67  137.25 1766.96  144.73 1768.33  151.13 1768.98
  175.89 1769.35  188.88 1770.11  202.97 1772.81  208.32 1774.33  211.72 1775.69
  224.03 1781.51  236.51 1788.29   243.5 1792.21  251.69 1797.84   260.5 1803.02
   266.5 1806.03  275.78 1809.82  284.07 1813.49  289.22 1816.02  292.09 1816.84
#Mann= 3 , 0 , 0
       0     .08       0   80.45     .05       0  126.36    .065       0
Bank Sta=80.45,126.36
Exp/Cntr=0.3,0.1

Type RM Length L Ch R = 1 ,47806   ,191.8,221.75,217.73
BEGIN DESCRIPTION:
47728.02
END DESCRIPTION:
XS GIS Cut Line= 6
  896866.5885877  809897.7074031  896913.4640812  809936.7704851
  896935.3384239  809946.1447645  897032.2141709  809963.3324796
  897066.5885769  810016.4574927  897075.9638804  810057.0824425
#Sta/Elev= 27
       0 1802.12   14.69 1796.57   19.88 1794.87      28 1791.29   38.59  1787.2
   41.76 1785.81   58.95 1776.15    61.8 1774.33   66.32 1772.97   73.38 1770.71
   83.15 1766.37   89.66 1765.15    92.8 1764.35  110.97 1764.17  135.47 1764.24
  143.69 1764.97  187.35 1769.01  223.82 1775.59  233.82 1781.21  236.23 1783.02
  244.63 1788.22   247.3 1790.09  253.25 1793.92  256.48 1795.74  263.23 1800.32
  278.98 1808.42  288.99 1812.95
#Mann= 3 , 0 , 0
       0    .075       0   89.66     .05       0  143.69     .07       0
Bank Sta=89.66,143.69
Exp/Cntr=0.3,0.1

Type RM Length L Ch R = 1 ,47584   ,324.93,291.02,243.91
BEGIN DESCRIPTION:
47506.27
END DESCRIPTION:
XS GIS Cut Line= 6
  896732.2136749  810064.8948541  896794.7139916   810085.207329
  896840.0265932  810110.2074557  896897.8392581  810157.0829492
  896927.5260124  810175.8325321  896999.4016326  810193.0202473
#Sta/Elev= 30
       0 1816.34    8.09 1810.06   13.38 1807.12   27.75  1797.3   40.51 1785.05
   46.67 1780.54    47.8  1779.8   50.26 1778.51   69.37 1774.29   81.76 1770.45
   94.26 1769.89  103.12 1769.34  113.14 1769.09  122.68 1768.65  128.95 1768.23
  152.83 1764.24  157.26 1763.75  160.72 1763.37  165.74 1762.45  173.17 1762.15
  189.39 1762.12  192.77  1762.2  204.32 1763.81  217.73 1771.38  227.46 1775.87
  254.64 1788.88  260.26 1792.59  274.37 1799.35  298.42 1807.26  301.37 1808.08
#Mann= 3 , 0 , 0
       0    .075       0  157.26     .05       0  204.32    .075       0
Bank Sta=157.26,204.32
Exp/Cntr=0.3,0.1

Type RM Length L Ch R = 1 ,47293   ,432.51,428.27,284.13
BEGIN DESCRIPTION:
47215.25
END DESCRIPTION:
XS GIS Cut Line= 6
  896566.5891159  810357.0829385  896657.2143191  810357.0829385
  896715.0259598  810372.7077616  896761.9014534    810402.39554
  896815.0264665  810414.8956034  896944.7137275  810408.6450596
#Sta/Elev= 30
       0 1821.92   12.67 1810.03   26.33 1798.02   33.79 1790.74   37.06 1787.97
   47.37 1781.37   65.28 1769.32   78.12 1767.61   96.77 1765.86  112.94 1762.81
  119.07 1761.87  133.14 1760.44  136.36 1760.29  161.01 1761.38  163.51 1761.57
   168.9 1762.51  189.46 1765.31  214.51 1765.27  245.98 1765.96  256.85 1766.69
  273.38 1768.63  307.06 1771.95  341.14 1773.17  351.14 1775.02  366.34 1778.29
  372.85 1781.02  375.94 1781.83  379.37 1783.02  386.12 1785.98  390.69 1787.66
#Mann= 3 , 0 , 0
       0    .075       0  112.94     .05       0   168.9     .07       0
Bank Sta=112.94,168.9
Exp/Cntr=0.3,0.1

Type RM Length L Ch R = 1 ,46865   ,280.07,242.29,130.45
BEGIN DESCRIPTION:
46786.98
END DESCRIPTION:
XS GIS Cut Line= 6
  896565.0262239  810786.7696712  896716.5888518   810791.457323
  896757.2138016  810782.0830436  896796.2758594  810764.8953285
  896921.2764928  810666.4577138  897005.6511522  810622.7080042
#Sta/Elev= 30
       0 1825.06    5.64 1820.33    20.8 1808.01   40.47 1790.09   72.85 1767.21
   76.36  1763.9   82.64 1761.17   88.61 1760.36  102.86  1758.6  125.71 1758.63
  132.23 1758.41  143.011760.047  152.14 1761.43  181.08 1764.94  192.96 1765.48
  206.74 1766.45  234.37 1767.98  266.17 1768.63  306.49 1767.79   337.8  1768.4
   347.7 1770.67  367.21 1774.52  375.52 1775.74  390.86  1783.2  391.46 1783.36
  408.88 1786.72  434.56 1793.93  454.09 1797.66  461.78 1799.78  490.86 1806.27
#Mann= 3 , 0 , 0
       0    .075       0   88.61     .05       0  143.01     .07       0
Bank Sta=88.61,143.01
Exp/Cntr=0.3,0.1

Type RM Length L Ch R = 1 ,46623   ,263.16,244.53,95.3
BEGIN DESCRIPTION:
46544.69
END DESCRIPTION:
XS GIS Cut Line= 6
  896644.7142557  811077.3948636   896713.464092  811024.2698504
  896791.5892318  810971.1448373  896836.9008092  810925.8322357
  896983.7768095   810736.770442  897032.2141709   810661.770062
#Sta/Elev= 30
       0 1828.21    2.16 1826.41    29.1 1798.25   38.17 1790.87   60.95 1771.38
   61.98 1770.33   68.22 1761.88   70.761759.744   74.87 1756.15   75.53 1756.05
  102.31    1757  114.42 1758.66  143.06 1762.02  157.29 1761.03  170.56 1759.42
  178.01 1761.84  196.64 1764.53  330.81 1766.83  362.39 1766.81  400.71 1766.16
  446.13 1766.47  459.86 1767.37  488.75 1770.21  491.49 1771.01  503.51    1776
  505.97 1777.47  518.95 1783.71  543.56 1794.39  555.57    1799  574.13 1804.61
#Mann= 3 , 0 , 0
       0     .07       0   70.76     .05       0  114.42     .07       0
#XS Ineff= 2 , 0
       0                  362.39       0    1772
Permanent Ineff=
       F       F
Bank Sta=70.76,114.42
Exp/Cntr=0.3,0.1

Type RM Length L Ch R = 1 ,46378   ,204.95,234.51,178.12
BEGIN DESCRIPTION:
46300.16
END DESCRIPTION:
XS GIS Cut Line= 6
  896908.7764295   811144.582832  896952.5261391  811068.0205842
  896949.4013793  810949.2704946  896968.1509622  810894.5825895
  897038.4636904  810811.7697979  897122.8383498  810703.9579038
#Sta/Elev= 30
       0 1794.99     4.3 1791.62   18.64 1782.42    25.7 1777.03   46.93 1761.81
   65.25 1759.65    74.1 1758.15   88.19 1757.12   97.11 1755.84  130.67 1755.46
  137.99 1756.41  146.63 1757.52  155.73 1758.11  176.09 1761.62  201.89 1764.39
  211.08 1764.94  270.86 1766.64  302.12 1768.21  329.18 1767.93  333.16 1767.43
  391.06 1768.24  404.89 1768.88  418.93 1770.71  423.66 1772.98  441.47 1779.31
  457.38 1786.21  462.41 1787.94  470.34 1791.89  487.98 1799.61  510.52  1810.2
#Mann= 3 , 0 , 0
       0    .065       0   88.19     .05       0  137.99     .07       0
Bank Sta=88.19,137.99
Exp/Cntr=0.3,0.1

Type RM Length L Ch R = 1 ,46144   ,80.73,167.35,280.51
BEGIN DESCRIPTION:
46065.65
END DESCRIPTION:
XS GIS Cut Line= 6
  897071.2762287  811233.6451432  897141.5889569  811150.8323516
  897168.1509514   811108.645534  897180.6510147  811066.4576922
  897185.3386665  810957.0829062  897208.7759012  810725.8322465
#Sta/Elev= 30
       0 1790.48    2.52 1789.68   10.36 1784.58   21.26 1778.56   31.47 1772.28
   43.07 1767.61   54.59 1764.51   94.08 1760.94   158.5 1758.11  173.92 1757.96
  230.64 1758.99  240.75 1755.78  246.91 1753.82  279.75 1753.41  287.65 1755.84
  300.68 1760.13  309.02 1762.62  311.07  1762.8  328.22  1768.1  337.57 1769.81
  383.46 1773.84  421.38 1774.47  449.37 1780.87  459.19 1781.68  463.24 1782.57
  477.56 1783.44   488.4 1784.72  494.35 1787.66  508.02 1796.29  544.86 1812.22
#Mann= 3 , 0 , 0
       0     .06       0  240.75     .05       0  287.65    .075       0
Bank Sta=240.75,287.65
Exp/Cntr=0.3,0.1

Type RM Length L Ch R = 1 ,45976   ,242.96,387.49,429.36
BEGIN DESCRIPTION:
45898.30
END DESCRIPTION:
XS GIS Cut Line= 6
  897118.1517222  811268.0205734  897185.3386665  811221.1450799
  897236.9018119  811168.0200667  897300.9639964  811077.3948636
   897382.213896  811039.8946736  897425.9636056  811008.6450273
#Sta/Elev= 30
       0 1784.95    5.24 1782.02   13.15  1778.7   20.36 1774.52   45.43 1766.96
   57.35 1765.37   66.71 1764.62   76.75 1764.66   83.55 1763.78  110.61 1762.32
   141.6 1760.33  150.26 1759.86  179.72 1758.76  193.69 1758.01  205.71 1757.05
   215.8 1757.61   233.8 1757.78  263.86 1757.69  267.45 1757.04  276.32 1755.05
  280.96 1754.22  290.41 1753.38  300.01 1753.01  302.22 1755.07  306.14 1757.57
  353.92 1787.97  362.11 1792.42  370.31 1792.51  374.47 1793.14   410.7 1822.97
#Mann= 3 , 0 , 0
       0    .055       0  267.45     .05       0  306.14    .085       0
Bank Sta=267.45,306.14
Exp/Cntr=0.3,0.1

Type RM Length L Ch R = 1 ,45589   ,200.88,247.92,275.68
BEGIN DESCRIPTION:
45510.81
END DESCRIPTION:
XS GIS Cut Line= 6
   897249.400851  811444.5823038  897349.4013577   811407.083138
  897424.4017378   811403.957354  897532.2136318  811397.7078344
  897568.1509299  811397.7078344  897633.7760064  811402.3954862
#Sta/Elev= 30
       0 1774.55    2.36  1773.7    9.54 1772.09   16.76 1771.25   25.49 1769.44
   29.48 1768.96    38.9 1767.14   68.03 1763.26   75.47 1762.95   80.65 1762.46
   96.48 1761.96  114.29 1761.53  133.52 1761.47  156.26 1760.97  172.24 1760.78
  195.29 1759.87  233.45 1754.82  239.81 1753.45  250.18 1750.63  268.38 1751.32
  277.26 1751.25  283.01 1752.08  300.48 1755.48  304.01 1756.28  337.64 1778.28
  343.78 1781.47  357.31 1794.74  382.61 1821.81  386.52 1826.49  391.59 1831.79
#Mann= 3 , 0 , 0
       0     .06       0  239.81     .05       0  300.48     .07       0
Bank Sta=239.81,300.48
Exp/Cntr=0.3,0.1

Type RM Length L Ch R = 1 ,45341   ,123.62,180.96,242.03
BEGIN DESCRIPTION:
45262.89
END DESCRIPTION:
XS GIS Cut Line= 6
  897271.2762179  811635.2080137  897327.5259908  811616.4574066
  897394.7139593  811614.8955388  897452.5266242  811636.7698815
  897494.7134418  811660.2081403  897582.2138852  811710.2073695
#Sta/Elev= 30
       0 1787.36   12.04 1786.79   30.53  1784.8   33.54 1783.49   62.01 1764.23
   72.19 1761.07   74.37  1759.8   77.27 1759.23   81.24 1759.03  106.25 1756.16
  122.01 1755.39  131.67 1755.34  144.19 1754.63   154.6 1753.35  159.27 1752.08
  167.16 1750.49  173.62 1749.82   187.8 1749.15  198.98 1749.59   210.6  1751.3
  215.431752.473  228.76 1755.81  233.34 1758.57   246.6 1768.16  253.54 1775.01
  260.24  1780.5     283 1801.68  300.04 1816.93  310.96  1825.2  337.35 1848.91
#Mann= 3 , 0 , 0
       0     .06       0  159.27     .05       0  215.43     .07       0
Bank Sta=159.27,215.43
Exp/Cntr=0.5,0.3

Type RM Length L Ch R = 1 ,45160   ,76.42,73.71,54.79
BEGIN DESCRIPTION:
45081.94
END DESCRIPTION:
XS GIS Cut Line= 6
  897280.6515215  811689.8948946  897333.7765346  811728.9579766
  897393.1510673  811882.0824723  897408.7758904   811943.019897
  897408.7758904  811972.7076754  897396.2758271  812044.5822715
#Sta/Elev= 30
       0 1785.74    20.7 1785.14   27.07 1784.45   35.22 1782.43   54.55 1772.65
   59.67 1769.11   68.47 1764.28   76.67 1758.96   88.42 1753.99   95.55 1752.28
  113.03 1749.45   142.1 1748.35  164.93    1749  167.11 1749.53  177.25 1750.32
  180.85 1752.46  190.61 1758.71  200.15 1764.21  204.23 1765.52  216.43 1771.02
  236.03 1776.54  246.23 1777.56  278.86 1776.86  308.58    1777  324.37 1776.25
  351.68 1813.22  371.09 1826.78   378.4 1831.19  381.34 1833.51  395.81 1842.26
#Mann= 3 , 0 , 0
       0    .055       0   95.55     .05       0  180.85     .06       0
Bank Sta=95.55,180.85
Exp/Cntr=0.5,0.3

Type RM Length L Ch R = 3 ,45132   ,,,
BEGIN DESCRIPTION:
45051.9  FBSTR_1286  No Photo
END DESCRIPTION:
Bridge Culvert--1,0,-1,-1, 0
Deck Dist Width WeirC Skew NumUp NumDn MinLoCord MaxHiCord MaxSubmerge Is_Ogee
12,37,2.6,0, 5, 5, , , 0.95, 0, 0,0,,
   33.36    41.5     135   228.5  330.52
 1782.84 1784.49 1784.49 1784.49 1784.59
         1781.49 1781.49 1781.49
   17.41   35.25     129   222.5  288.24
 1782.61 1784.49 1784.49 1784.49 1784.58
         1781.49 1781.49 1781.49
BR Coef=-1 , 0 , 0 ,, 0 ,,,0.8,0,,0,
WSPro=,,,, 1 ,,,, 0 ,,,, 0 ,,,,-1 ,-1 ,-1 , 0 , 0 , 0 , 0 , 0
BC Design=,, 0 ,, 0 ,,,,,,

Type RM Length L Ch R = 1 ,45086   ,153.43,171.52,217
BEGIN DESCRIPTION:
45008.22
END DESCRIPTION:
XS GIS Cut Line= 6
  897274.4009777  811707.0826097  897277.5267617  811783.6448576
  897313.4640597  811857.0823456  897349.4013577  811911.7702507
  897361.9014211  811939.8951372   897363.464313  812025.8326886
#Sta/Elev= 30
       0 1784.81   12.73 1784.64   17.41 1782.61   32.23 1778.24   38.22 1776.05
   52.13 1768.55   65.42 1763.22    78.4  1756.2   86.94 1754.25   90.73 1753.83
  102.27 1751.01  115.23 1748.27  123.08 1747.93  155.43 1748.66  159.89  1749.1
  164.63 1750.11  168.22 1750.36  178.04  1755.4  186.17 1759.18  195.64 1766.03
  215.11 1773.45  218.99 1775.57  220.95 1775.64  234.08 1778.46   251.8 1778.35
  279.69  1777.4  288.24 1784.58  307.76 1810.66  320.94 1819.25  340.85    1830
#Mann= 3 , 0 , 0
       0     .06       0  102.27     .05       0  168.22    .055       0
Bank Sta=102.27,168.22
Exp/Cntr=0.5,0.3

Type RM Length L Ch R = 1 ,44915   ,129.27,197.09,240.73
BEGIN DESCRIPTION:
44836.70
END DESCRIPTION:
XS GIS Cut Line= 5
  897115.0259383   811739.895148  897144.7137167  811871.1453009
  897144.7137167  811903.9578392  897141.5889569  811966.4571317
  897135.3384132  812027.3955806
#Sta/Elev= 30
       0 1773.45    6.38 1773.03    8.57 1772.56   33.55 1768.88   58.17 1764.15
   76.14 1760.99   83.84 1759.15    91.7 1757.92  100.33 1756.02  120.64  1752.5
  131.88 1750.35  137.21 1749.08  146.11 1746.74  157.47 1745.66  159.95 1745.14
  167.22 1745.79  173.13 1745.72  176.62    1746  183.54 1748.66  190.64 1754.38
  202.67 1763.42  218.05 1777.87  229.33 1785.43  240.04 1785.83  248.75 1787.22
     250  1787.2  260.48 1794.49  263.23 1796.83  270.47 1805.87  291.21 1829.28
#Mann= 3 , 0 , 0
       0    .055       0  137.21     .05       0  183.54    .055       0
Bank Sta=137.21,183.54
Exp/Cntr=0.3,0.1

Type RM Length L Ch R = 1 ,44718   ,428.13,420.27,372.24
BEGIN DESCRIPTION:
44639.62
END DESCRIPTION:
XS GIS Cut Line= 6
  897049.4008618  811697.7073062  897035.3389306    811741.45804
  896983.7768095  811802.3954647  896936.9013159  811841.4575225
  896919.7136008  811866.4576492  896896.2763661  811925.8321819
#Sta/Elev= 30
       0 1775.49    17.2 1773.11   33.21 1771.18   43.19 1769.66   45.96 1768.88
   53.97 1766.16   69.15 1759.96   77.71 1755.26   88.86 1751.21   98.94 1747.34
  102.49 1746.87  112.89  1746.3  132.31 1745.92  145.23 1745.29  152.78 1746.06
  172.96 1747.22   178.6    1748  184.23 1748.56   191.4 1748.74  204.87  1752.2
  210.97 1755.36  218.34 1758.88  221.46 1760.79  233.02 1769.96  244.18 1778.57
  256.51 1787.24  260.51 1789.55  267.21 1793.09  280.13 1799.27  281.46 1799.22
#Mann= 3 , 0 , 0
       0    .065       0   98.94     .05       0   178.6     .06       0
Bank Sta=98.94,178.6
Exp/Cntr=0.3,0.1

Type RM Length L Ch R = 1 ,44297   ,506.25,435.48,273.32
BEGIN DESCRIPTION:
44219.35
END DESCRIPTION:
XS GIS Cut Line= 6
  896668.1514904   811535.207507  896646.2761235   811574.270589
  896605.6511737  811625.8327101  896574.4015275  811714.8950213
  896572.8386355  811747.7075595  896580.6510471  811799.2696807
#Sta/Elev= 30
       0 1785.26    4.21  1782.5   30.35 1764.35   38.18 1760.18   44.77 1755.54
   49.24 1752.48   79.18  1745.9   84.81 1744.67   93.01 1742.61   95.42 1742.57
  107.78  1742.7  117.55  1742.4  124.39 1742.77  131.81 1744.22  134.72 1744.24
  138.19 1745.01  143.29 1745.36  153.49 1746.21  166.61 1746.37  175.59 1746.67
  181.33 1747.09  189.41 1747.98   203.3 1750.58  206.96 1751.44  217.82 1754.54
  231.22 1758.76  235.52 1759.51  245.19 1761.45  273.83 1765.63  289.88 1767.12
#Mann= 3 , 0 , 0
       0     .09       0   79.18     .05       0  131.81    .055       0
#Block Obstruct= 1 ,-1
  275.49  289.881777.124
Bank Sta=79.18,131.81
Exp/Cntr=0.3,0.1

Type RM Length L Ch R = 1 ,43862   ,242.49,186.83,20.05
BEGIN DESCRIPTION:
43783.87
END DESCRIPTION:
XS GIS Cut Line= 6
  896157.2138339  811503.9578607  896207.2140872  811619.5821664
  896260.3391004  811688.3330268  896315.0259813  811736.7703882
  896358.7767151  811761.7705149  896444.7142665  811802.3954647
#Sta/Elev= 30
       0 1796.72    3.08 1793.35   21.76 1774.83   36.05    1761   51.05 1750.42
   57.03 1744.13   61.68 1743.28   67.04 1741.04   70.09 1739.76   79.68 1740.11
   103.6 1740.37  108.59  1740.6  129.16 1741.78  134.82 1742.37  140.75 1742.54
  143.94 1743.18  153.18 1744.14  166.98 1746.25  175.16 1746.88  184.35 1748.05
  199.42 1749.23   220.9 1751.47  251.03 1753.91  276.93 1755.22  322.45 1755.99
  342.86 1755.99  362.53 1756.44  389.23 1757.76  404.04 1759.09  431.44 1760.52
#Mann= 3 , 0 , 0
       0    .085       0   67.04     .05       0  108.59     .05       0
#Block Obstruct= 1 ,-1
  418.85  431.441770.525
Bank Sta=67.04,108.59
Exp/Cntr=0.3,0.1

Type RM Length L Ch R = 1 ,43675   ,245.43,220.85,113.92
BEGIN DESCRIPTION:
43597.04
END DESCRIPTION:
XS GIS Cut Line= 6
  895988.4634909  811725.8321926   896043.151396  811730.5198444
  896241.5884933    811741.45804  896280.6515753    811741.45804
  896321.2765251  811758.6447309  896416.5883559   811811.769744
#Sta/Elev= 30
       0 1809.74   22.32 1784.79   50.69 1755.06   58.66 1748.62   63.46 1743.77
   66.48 1743.49   77.27 1741.42    83.3 1739.97   90.22  1738.3  102.54    1739
  108.53 1739.78  120.09 1740.99  131.61 1741.77  134.88 1741.79  152.53 1740.94
  177.79 1745.36  186.24 1746.22   203.2 1747.54  212.79 1747.88  240.76 1749.82
   249.6  1750.6  255.67 1750.85  264.52 1751.87  301.16 1754.54  309.23 1754.81
  344.22 1755.38  370.45 1755.52  412.23 1757.18  433.86 1758.44  445.93 1758.96
#Mann= 3 , 0 , 0
       0    .075       0    83.3     .05       0  108.53     .05       0
Bank Sta=83.3,108.53
Exp/Cntr=0.3,0.1

Type RM Length L Ch R = 1 ,43454   ,195.2,179.61,75.95
BEGIN DESCRIPTION:
43376.19
END DESCRIPTION:
XS GIS Cut Line= 6
  896019.7141614  811994.5830423  896130.6508152  811936.7703774
  896182.2139606  811894.5825356  896221.2760184  811877.3948205
  896336.9013482  811857.0823456  896440.0266147   811850.832826
#Sta/Elev= 30
       0 1812.55   10.59 1801.52    16.1  1793.9   34.05 1769.78   37.77 1764.63
   67.57 1740.94   68.97 1739.94   73.43 1736.76   94.47 1736.73  118.741738.004
  131.46 1738.65  139.93 1738.63  145.06 1739.05   158.9 1737.47  166.45 1736.42
  175.04 1737.85  185.09  1741.9  195.21 1742.62  233.93 1746.84  262.77 1749.56
   269.5 1750.04  276.98 1750.37  294.09 1751.57  310.34 1752.86  326.96 1754.42
  352.47 1756.11  398.16 1758.19  422.29 1758.96  431.37  1759.5  456.17 1760.58
#Mann= 3 , 0 , 0
       0     .07       0   68.97     .04       0  118.74     .06       0
#Block Obstruct= 1 ,-1
  445.26  456.171770.575
Bank Sta=68.97,118.74
Exp/Cntr=0.3,0.1

Type RM Length L Ch R = 1 ,43274   ,416.42,395.66,377.55
BEGIN DESCRIPTION:
43196.57
END DESCRIPTION:
XS GIS Cut Line= 6
  896199.4016757  812107.0825882  896232.2142139  812052.3946831
  896265.0267522  811993.0201503  896358.7767151  811891.4577758
  896408.7759443  811868.0205411  896443.1513745  811863.3328894
#Sta/Elev= 28
       0 1798.18    20.4 1780.16   53.96 1745.23   60.74 1738.45    62.6 1736.59
   65.76 1736.33   88.78 1734.98   94.28 1734.96  111.18 1735.14  121.13 1735.35
  127.95 1735.78  137.36 1738.34  141.26 1739.36   144.6 1739.72     153 1740.89
  167.49 1742.59  181.18 1744.36  205.98  1748.2  229.91 1752.06  245.26 1754.03
  254.06 1755.05  274.12 1756.63   284.9 1757.27  311.33 1758.54  336.48 1759.37
  340.79 1759.63  347.49 1759.81  359.74 1760.38
#Mann= 3 , 0 , 0
       0     .07       0   60.74     .04       0  137.36    .065       0
#Block Obstruct= 1 ,-1
  344.52  359.741770.382
Bank Sta=60.74,137.36
Exp/Cntr=0.3,0.1

Type RM Length L Ch R = 1 ,42879   ,89.43,142.88,163.1
BEGIN DESCRIPTION:
42800.91
END DESCRIPTION:
XS GIS Cut Line= 6
  896611.9017175  812236.7698492  896613.4635853    812149.27043
  896633.7760602  812080.5205937  896649.4008833  812058.6452268
  896654.0885351  812039.8956439  896707.2135482  811991.4572584
#Sta/Elev= 30
       0 1766.32    7.06 1763.82   12.99 1760.21   20.08 1755.67   32.58 1749.62
   38.59 1747.09   41.68 1745.52   46.42 1743.46   50.28 1742.31   69.63 1737.14
   81.33 1735.97   90.67 1734.69  100.29 1732.98  111.97 1731.65  120.83 1731.89
  122.62 1731.84  133.46 1732.34  145.36 1733.66  154.41 1734.88  167.63 1737.52
  179.61 1739.14  186.29 1740.62  190.95 1741.71  201.81 1744.82  218.39 1748.11
  236.31 1752.19  257.06 1757.24  263.73 1758.75  273.48  1761.3  277.54 1762.48
#Mann= 3 , 0 , 0
       0    .075       0   90.67     .05       0  154.41     .06       0
#Block Obstruct= 1 ,-1
  227.79  267.581769.758
Bank Sta=90.67,154.41
Exp/Cntr=0.3,0.1

Type RM Length L Ch R = 1 ,42736   ,65.25,141.79,169.79
BEGIN DESCRIPTION:
42658.03
END DESCRIPTION:
XS GIS Cut Line= 6
  896654.0885351   812260.208108  896699.4011367  812225.8326778
  896740.0260865  812171.1447727  896772.8386247  812133.6456069
  896821.2759861  812100.8330686  896852.5266565  812093.0196329
#Sta/Elev= 30
       0 1768.29   15.24 1764.84   22.63 1762.59   24.56 1761.68   25.76 1761.41
   56.88 1752.63   60.53  1751.7   65.84 1748.92   74.02 1743.78   83.48 1738.64
   94.04 1736.47  103.66 1735.66  107.49  1735.5  109.55 1735.14  114.16 1734.04
   131.6 1730.26   132.9 1730.07  141.88  1730.3  157.68 1729.67  158.88 1729.81
  172.92 1732.91  174.85  1733.5  179.96 1734.76  189.39 1739.06     204 1746.79
  218.67 1752.86  233.43 1762.18  249.97 1772.39  262.34 1781.59  265.64 1783.63
#Mann= 3 , 0 , 0
       0     .07       0  114.16     .05       0  174.85    .075       0
Bank Sta=114.16,174.85
Exp/Cntr=0.3,0.1

Type RM Length L Ch R = 1 ,42594   ,27.95,81.68,107.54
BEGIN DESCRIPTION:
42516.24
END DESCRIPTION:
XS GIS Cut Line= 6
  896660.3390789  812282.0824507   896710.338308  812282.0824507
  896758.7766936   812277.394799  896802.5264032  812272.7071472
   896844.714245  812258.6452161  896911.9011892  812255.5204563
#Sta/Elev= 30
       0 1766.36   21.98 1758.69   27.08 1757.89   32.86 1755.77   38.36  1754.1
   43.43  1753.1   52.81 1751.58   60.74 1750.61   65.62  1750.5   70.89 1750.68
    79.3 1747.85  107.78 1739.84  119.14 1737.18  123.86 1735.92  134.22 1734.07
  142.66 1732.74  146.57 1732.06  160.34 1730.78  166.99 1729.89  169.18 1729.84
  186.42 1730.47  194.28 1730.46  198.66 1731.34  205.74 1733.73  213.47 1737.51
  226.71 1744.55  230.34 1748.42  234.51 1754.25  248.45 1775.29  254.47 1785.61
#Mann= 3 , 0 , 0
       0     .07       0  142.66    .045       0  205.74    .075       0
Bank Sta=142.66,205.74
Exp/Cntr=0.3,0.1

Type RM Length L Ch R = 1 ,42512   ,52.74,140.83,211.8
XS GIS Cut Line= 6
  896655.6514271  812296.1454061  896744.7137383  812313.3331212
  896799.4016434  812332.0827041  896836.9008092  812346.1446352
  896868.1514797  812357.0828308  896929.0889044  812366.4581343
#Sta/Elev= 30
       0 1764.85    2.97  1764.3   14.79 1761.28   23.21  1758.2   40.58 1755.22
   52.67 1752.18   67.08 1749.34   72.93 1747.91   81.33 1747.25      85 1746.71
  102.58  1743.3  113.24 1740.85  121.02  1739.5  126.78 1737.96  146.32 1731.74
  150.77 1730.81  153.54 1730.51  167.87    1730  179.28 1728.92  182.92 1728.86
  186.09 1728.92  197.32 1729.89  205.69 1733.18  206.35 1733.42  225.67 1747.55
   226.7 1748.88  256.14 1781.04  259.31 1785.05  276.64 1805.61  283.33 1812.67
#Mann= 3 , 0 , 0
       0     .07       0  146.32    .045       0  205.69    .075       0
Bank Sta=146.32,205.69
Exp/Cntr=0.3,0.1

Type RM Length L Ch R = 1 ,42372   ,176.6,216.38,220.85
XS GIS Cut Line= 6
  896652.5266673  812311.7702292  896685.3392055  812349.2704192
  896718.1517438   812388.332477  896724.4012634  812436.7698384
  896727.5260231   812483.645332  896727.5260231  812514.8949782
#Sta/Elev= 30
       0 1761.07    2.77 1760.26    11.9  1758.1   15.81 1757.02   36.51 1750.68
   50.65 1744.63   53.19 1743.82   58.99 1742.35   68.01 1740.47   73.44 1738.89
   88.56 1737.45  100.84 1736.07  103.67 1735.63  109.16    1732  119.62 1729.24
  122.99 1729.17  132.16 1728.12   146.8 1728.97  153.24 1729.22  156.65 1729.19
  165.34 1728.82  169.07 1729.02  171.14 1729.78  181.21 1733.13  191.21 1735.65
  198.73 1741.79  201.47 1743.89  205.67 1746.83  217.13 1756.61  227.91 1767.47
#Mann= 3 , 0 , 0
       0     .07       0  119.62    .045       0  171.14    .075       0
Bank Sta=119.62,171.14
Exp/Cntr=0.3,0.1

Type RM Length L Ch R = 1 ,42155   ,432.79,422.4,415.76
BEGIN DESCRIPTION:
42077.35
END DESCRIPTION:
XS GIS Cut Line= 3
  896505.6516912  812332.0827041   896507.213559  812499.2701551
  896513.4641028  812539.8951049
#Sta/Elev= 20
       0 1759.24    5.45 1756.24   25.26 1746.32   28.05 1744.45   37.65 1738.67
   49.68 1733.84   57.36 1729.73   62.34 1727.06   74.81 1726.68   84.49 1726.79
   92.55  1726.7  111.74 1726.86  121.38 1727.02  122.97 1726.95   141.4 1729.56
   155.3 1731.21  163.66 1734.14  168.18 1738.55  179.45 1743.17   208.3 1764.58
#Mann= 3 , 0 , 0
       0     .08       0   57.36     .05       0   141.4    .075       0
Bank Sta=57.36,141.4
Exp/Cntr=0.3,0.1

Type RM Length L Ch R = 1 ,41733   ,428.93,430.87,409.68
BEGIN DESCRIPTION:
41654.94
END DESCRIPTION:
XS GIS Cut Line= 4
   896061.900979  812322.7074006  896085.3392378  812393.0201288
  896083.7763459  812450.8327937  896102.5259288  812566.4581236
#Sta/Elev= 29
       0 1783.03   37.28 1752.17   61.58 1731.35   65.95 1728.96   71.48 1723.94
   77.51 1723.57   83.19 1723.44   99.03 1722.54  106.12 1722.73  110.87 1723.12
  114.79 1723.24  121.66 1723.31  129.72    1724  139.17 1726.79  145.67 1729.29
  150.94 1730.38  159.35 1731.08  168.61 1732.01  179.59 1732.71  187.57  1733.4
  195.82 1734.45  199.17 1734.96  205.65 1736.12  213.99 1737.16  225.47 1738.83
  235.76 1740.73   243.9 1742.74  247.72  1743.4  249.09 1743.76
#Mann= 3 , 0 , 0
       0    .085       0   65.95     .05       0  139.17    .055       0
Bank Sta=65.95,139.17
Exp/Cntr=0.3,0.1

Type RM Length L Ch R = 1 ,41302   ,231.36,267.05,289.9
BEGIN DESCRIPTION:
41224.07
END DESCRIPTION:
XS GIS Cut Line= 4
  895654.0885889  812393.0201288  895654.0885889  812450.8327937
   895672.839196  812539.8951049  895716.5889056  812664.8947141
#Sta/Elev= 30
       0 1773.46    8.28 1766.07   24.56 1752.42   40.13  1739.2   54.86 1727.47
   59.77 1723.97   62.29 1723.71   70.06 1721.88   73.44 1721.27   84.43 1720.45
   99.64  1720.3   103.8 1720.68  109.49 1720.93  122.06 1723.36   131.7 1725.28
  137.87 1727.63  144.15  1729.3  147.97 1729.74  153.28 1730.03  167.18 1731.56
  182.77 1733.67  188.01 1734.59  195.09 1735.09   204.7 1736.58  216.58 1738.21
  223.37 1739.02  242.39 1741.79  251.68 1743.38  261.08 1744.79  281.26 1748.57
#Mann= 3 , 0 , 0
       0    .085       0   62.29     .05       0  122.06     .06       0
Bank Sta=62.29,122.06
Exp/Cntr=0.3,0.1

Type RM Length L Ch R = 1 ,41035   ,245.22,268.09,324.51
BEGIN DESCRIPTION:
40957.01
END DESCRIPTION:
XS GIS Cut Line= 6
  895482.2134862  812377.3953057  895408.7759981  812461.7699651
  895402.5264785  812486.7700918  895402.5264785  812508.6454586
  895415.0265419  812608.6449412  895418.1513017  812750.8322655
#Sta/Elev= 30
       0 1768.34   20.98 1763.43   37.46 1755.19   46.07  1751.1   62.34 1743.86
   70.86 1739.86   77.34 1737.35   84.22 1733.86   96.38 1731.75  109.51 1730.61
  144.99 1728.91  172.71  1728.3  194.12 1721.61  204.78 1719.86  220.29 1719.46
   229.6  1719.4  241.58 1719.64  250.79 1720.94  260.38 1724.65  266.74 1727.98
  278.41 1729.67  298.55 1731.22  309.65 1732.61  334.46  1736.1  346.94 1738.06
  357.15 1739.52  368.47 1741.68  383.88 1746.92     389 1748.53  402.57 1752.32
#Mann= 3 , 0 , 0
       0    .075       0  194.12     .05       0  250.79     .06       0
Bank Sta=194.12,250.79
Exp/Cntr=0.3,0.1

Type RM Length L Ch R = 1 ,40767   ,128.85,166.55,187.32
BEGIN DESCRIPTION:
40688.92
END DESCRIPTION:
XS GIS Cut Line= 6
  895199.6956679  812403.0314454  895199.6956679  812434.2810917
  895191.8832564  812471.7812817  895162.1954779  812526.4691868
  895120.0086603  812582.7189597  895082.5084703  812628.0315613
#Sta/Elev= 28
       0 1734.66    7.42 1734.13   31.25 1733.27   41.12 1732.83   54.56 1731.96
   69.74 1730.59   83.79 1728.71   92.01 1727.24   97.85 1726.32   108.3  1724.4
  111.79 1723.69  125.84 1720.54  138.68 1718.58  141.92 1718.21   150.5  1717.7
   172.9 1717.25  180.65 1717.31  186.66 1717.91  193.35  1718.9  195.76 1719.87
  207.87 1725.79  210.84 1727.78  215.52 1729.94  221.48 1734.25  234.89 1745.71
  252.69 1758.31  258.36    1764  260.91 1766.93
#Mann= 3 , 0 , 0
       0     .06       0  141.92     .05       0  186.66     .07       0
Bank Sta=141.92,186.66
Exp/Cntr=0.3,0.1

Type RM Length L Ch R = 1 ,40600   ,148.31,151.03,144.61
BEGIN DESCRIPTION:
40522.37
END DESCRIPTION:
XS GIS Cut Line= 6
  895135.6334834  812323.3444378  895101.2580532  812382.7189705
  895074.6960587  812407.7190972  895032.5082169  812429.5944641
  894985.6337475  812460.8441103  894930.9458424  812463.9688701
#Sta/Elev= 30
       0  1758.1   25.71 1746.26   26.41 1745.83   27.79 1745.33   48.19 1736.92
   71.32 1725.29   75.22 1724.43   81.34 1720.34   89.88 1720.26   97.69 1719.17
  109.81 1717.76  115.25 1717.47  123.08 1716.87  135.17 1716.74  144.49 1716.54
  162.97  1716.7  167.18 1716.83  180.88  1716.9  182.09 1717.36  188.23 1719.79
  195.39 1722.51  201.78 1727.47  208.97 1733.42  220.54 1742.28  221.25 1742.67
  235.51 1754.61  242.04 1760.93  244.36 1763.44  248.63 1766.74  263.75 1779.44
#Mann= 3 , 0 , 0
       0     .08       0  115.25     .05       0  182.09     .07       0
Bank Sta=115.25,182.09
Exp/Cntr=0.3,0.1

Type RM Length L Ch R = 1 ,40449   ,183.83,136.7,96.64
BEGIN DESCRIPTION:
40371.34
END DESCRIPTION:
XS GIS Cut Line= 6
  895062.1959954  812224.9068231  895007.5080903  812273.3441844
   894974.695552  812290.5318995  894948.1335575  812309.2814825
  894913.7581273  812337.4063689  894887.1961328   812373.343667
#Sta/Elev= 26
       0 1780.57   16.63 1766.52   40.13 1743.93   63.86 1721.33   70.681716.593
   72.44 1715.37   73.05 1715.35   83.28 1714.93   90.19 1714.57   97.78 1714.42
  104.06 1714.47  108.82 1714.47   110.1 1714.53  110.46 1714.55  111.67  1714.6
  116.72 1714.96   123.6 1715.45  138.93 1715.65  139.09 1715.66  139.45 1715.71
  157.78 1718.14  161.67 1718.52  206.21 1743.09  206.97 1743.38  211.15 1746.23
  231.71 1760.18
#Mann= 3 , 0 , 0
       0     .08       0   70.68     .05       0  116.72     .07       0
Bank Sta=70.68,116.72
Exp/Cntr=0.3,0.1

Type RM Length L Ch R = 1 ,40313   ,305.85,272.85,194.51
XS GIS Cut Line= 6
  894899.6961962  812090.5319103   894902.820956  812140.5311395
   894902.820956  812170.2189179  894890.3208926  812193.6561526
  894849.6959428  812271.7812924  894813.7586448  812326.4691976
#Sta/Elev= 28
       0 1760.11   16.13 1747.19    50.1 1720.96   55.73 1716.59   57.91 1715.45
    64.9 1714.92   73.91 1714.13   79.67 1713.89   83.05 1713.83   86.31 1713.59
   91.07 1713.74   98.43 1714.23  103.02 1714.53  106.35 1714.62  109.01 1714.69
  109.42 1714.71   113.4 1714.92  116.12 1715.08  122.99 1715.46  130.18 1715.83
  137.53 1716.37  151.92 1716.65  172.16  1716.7   176.6 1717.64   194.4 1726.89
   219.1 1739.74  220.85  1740.6  259.84 1762.01
#Mann= 3 , 0 , 0
       0     .08       0   57.91     .05       0  109.42     .07       0
Bank Sta=57.91,109.42
Exp/Cntr=0.3,0.1

Type RM Length L Ch R = 1 ,40040   ,429.28,417.63,411.32
BEGIN DESCRIPTION:
39961.79
END DESCRIPTION:
XS GIS Cut Line= 6
  894579.3832253  812128.0310762  894620.0081751  812193.6561526
  894635.6329983  812221.7810391  894660.6331249  812249.9069497
   894679.383732  812268.6565327  894687.1961436  812298.3443111
#Sta/Elev= 21
       0 1745.72   18.93 1736.24   42.97 1724.92   44.49 1724.02   49.25 1720.92
   54.33 1717.02   77.18 1712.13   80.61 1711.38   81.33 1711.32   88.94 1710.97
  101.61 1710.55  107.08 1710.95  117.59 1711.22  119.141712.155  145.67 1728.16
  162.37 1735.09   173.5 1740.12   183.4  1745.5  186.92 1746.98  193.19 1750.33
   204.2  1756.7
#Mann= 3 , 0 , 0
       0     .08       0   77.18    .055       0  119.14    .065       0
Bank Sta=77.18,119.14
Exp/Cntr=0.3,0.1

Type RM Length L Ch R = 1 ,39622   ,425.74,441.13,452.12
BEGIN DESCRIPTION:
39544.16
END DESCRIPTION:
XS GIS Cut Line= 3
  894254.3836269  812421.7810283  894310.6333998  812474.9060415
  894374.6955843   812540.531118
#Sta/Elev= 20
       0 1747.04   16.87 1736.45   29.59 1727.99   47.65 1715.14   51.93 1712.54
   67.88 1705.38   69.37 1704.51   71.63 1704.44   73.69 1704.37   92.06 1703.69
   93.65 1703.65   99.17 1703.79   101.7 1703.85  106.74 1703.91  106.85 1703.91
  111.47  1704.1  114.61 1704.43  157.14 1727.03  166.58 1732.27  169.08 1733.96
#Mann= 3 , 0 , 0
       0     .08       0   67.88     .05       0  106.74     .07       0
Bank Sta=67.88,106.74
Exp/Cntr=0.3,0.1

Type RM Length L Ch R = 1 ,39181   ,220.81,250.38,290.15
BEGIN DESCRIPTION:
39103.03
END DESCRIPTION:
XS GIS Cut Line= 5
  893937.1954158  812670.2194031  893957.5078907  812732.7186956
   893993.446213   812781.156057  894018.4463396  812813.9685952
  894049.6959859  812868.6565004
#Sta/Elev= 22
       0 1745.89   14.79 1739.47   31.36 1724.09   55.56 1710.05   60.91 1706.67
   65.15 1704.16   79.97 1702.37   85.18 1702.55   98.64 1702.41  114.56 1702.47
  123.25 1702.36  125.85  1702.4  133.33 1702.84  136.111703.128  146.38 1704.19
   152.2 1705.17  158.93 1706.54  164.13 1707.04  175.02 1710.91  176.02 1711.13
  217.79 1728.82  230.27 1735.93
#Mann= 3 , 0 , 0
       0     .08       0   79.97     .05       0  136.11    .075       0
Bank Sta=79.97,136.11
Exp/Cntr=0.3,0.1

Type RM Length L Ch R = 1 ,38931   ,97.67,172.5,219.6
BEGIN DESCRIPTION:
38852.65
END DESCRIPTION:
XS GIS Cut Line= 6
  893748.1336221  812734.2815876    893749.69549   812781.156057
  893757.5079015  812868.6565004  893773.1337488  812906.1566904
  893777.8203764  812928.0310331  893779.3832684    812987.40659
#Sta/Elev= 24
       0 1752.32   22.01 1734.72   37.64 1724.44   40.02 1722.96   44.03 1721.51
   51.99 1717.27   95.08 1708.22  109.74 1704.99  113.86 1704.57  137.16 1701.44
   146.1 1700.31  157.41 1700.22  159.84 1700.28   173.6 1699.64  177.16  1700.2
  182.231701.334  187.87 1702.67  194.98 1702.11  198.56 1702.63  203.55  1704.5
  233.46 1713.61  240.71 1718.35  251.26 1724.48  257.17 1728.16
#Mann= 3 , 0 , 0
       0    .085       0  137.16     .05       0  182.23    .075       0
Bank Sta=137.16,182.23
Exp/Cntr=0.3,0.1

Type RM Length L Ch R = 1 ,38758   ,107.12,152.03,169.78
BEGIN DESCRIPTION:
38680.15
END DESCRIPTION:
XS GIS Cut Line= 6
  893677.8208939  812732.7186956   893657.508419  812778.0312972
  893591.8833425  812904.5937984  893571.5708676  812920.2186215
  893562.1955641  812942.0939884  893559.0708043  812968.6559829
#Sta/Elev= 26
       0 1748.36   17.63 1734.51   43.85 1712.95   49.66 1708.92   50.53 1708.32
   60.47 1706.64   79.14 1705.17   96.68 1703.62  142.491699.892  146.21 1699.59
  148.74 1699.38  152.36 1699.41  164.63 1699.38  167.01 1699.39  176.97 1699.33
  180.93 1699.27  182.78 1699.27  189.18 1699.26  192.35 1699.29  196.67 1699.32
  197.74 1700.26  199.39 1701.71  217.98 1712.11  239.61 1726.17  241.78 1727.62
  268.52 1744.89
#Mann= 3 , 0 , 0
       0    .085       0  142.49     .05       0  197.74    .075       0
Bank Sta=142.49,197.74
Exp/Cntr=0.3,0.1

Type RM Length L Ch R = 1 ,38606   ,229.59,248.61,270.76
BEGIN DESCRIPTION:
38528.12
END DESCRIPTION:
XS GIS Cut Line= 6
  893588.7585827  812696.7813976  893554.3831525  812740.5311072
  893530.9459178  812759.2817143  893509.0705509  812768.6559937
  893423.1329995  812834.2810701  893391.8833533  812840.5316139
#Sta/Elev= 22
       0 1742.24    31.4 1722.01   48.98 1708.91    57.6 1708.19   85.65 1702.66
   101.2 1699.77  112.39 1697.96  122.97 1697.85  130.88 1697.96  141.67 1697.99
  154.89  1697.9   162.3  1698.2     172 1698.81  197.89 1710.55  199.63 1711.21
   201.4 1712.31  221.23 1726.51  228.25 1733.42  233.37 1737.89  241.21 1743.04
  248.73 1750.75  249.51 1751.47
#Mann= 3 , 0 , 0
       0    .085       0   101.2     .05       0   162.3    .075       0
Bank Sta=101.2,162.3
Exp/Cntr=0.3,0.1

Type RM Length L Ch R = 1 ,38357   ,439.78,445.07,444.95
BEGIN DESCRIPTION:
38279.51
END DESCRIPTION:
XS GIS Cut Line= 2
  893485.6333162  812529.5939466  893305.9458019  812587.4066115
#Sta/Elev= 26
       0 1734.89   14.81 1726.17   52.71 1702.76   83.681697.292    86.3 1696.83
   91.31 1695.96   92.44 1695.95   93.98 1695.97   99.74 1695.93  102.19 1695.92
  111.42 1696.11  114.22 1696.08   119.1 1695.97  121.45 1696.07  123.75 1696.11
  126.54 1696.17  129.34 1696.26  131.92 1696.21  139.58 1696.77  143.34 1697.31
   147.3 1697.91  164.29 1703.84  165.08 1704.14  165.72 1704.42  166.46 1704.98
  188.76 1720.37
#Mann= 3 , 0 , 0
       0    .085       0   83.68     .05       0  129.34    .075       0
Bank Sta=83.68,129.34
Exp/Cntr=0.3,0.1

Type RM Length L Ch R = 1 ,37912   ,437.26,420.45,415.28
BEGIN DESCRIPTION:
37834.44
END DESCRIPTION:
XS GIS Cut Line= 3
  893343.4459919  812115.5310128  893246.5712692  812138.9692717
  893160.6337178  812167.0941581
#Sta/Elev= 24
       0 1726.21   29.16 1708.39   45.14 1699.73   78.841694.733   80.88 1694.43
   86.23 1693.36   90.53 1693.37   94.13 1693.33   94.66 1693.32   97.82 1693.36
  101.32 1693.36  105.82 1693.24  118.16 1693.19  119.57 1693.19  123.71  1693.2
  127.31 1693.19  129.17 1693.26  140.75 1693.22  141.15 1693.22  148.24 1695.58
  154.78 1697.27  160.87 1698.63  164.72 1700.83  190.09  1721.2
#Mann= 3 , 0 , 0
       0    .085       0   78.84     .05       0  140.75     .07       0
Bank Sta=78.84,140.75
Exp/Cntr=0.3,0.1

Type RM Length L Ch R = 1 ,37492   ,416.84,427.84,431.23
BEGIN DESCRIPTION:
37414.00
END DESCRIPTION:
XS GIS Cut Line= 3
  893196.5710158  811699.9062112  893076.2580342  811754.5941163
  892991.8833748  811788.9685224
#Sta/Elev= 25
       0 1730.85   19.26 1711.34   26.52 1708.48   43.74 1702.99   93.12    1692
   93.94 1691.84   95.37 1691.54   95.81 1691.53   96.46 1691.53  107.44 1691.44
  109.85 1691.45  116.68 1691.54  117.81 1691.54  121.75 1691.59  126.88 1691.64
  127.44 1691.64  141.47 1691.73  144.42 1691.84  146.89 1692.24  152.19 1692.84
  160.53 1695.02  190.23 1702.41   199.7 1707.41  216.24 1723.17  223.27 1729.16
#Mann= 3 , 0 , 0
       0    .085       0   93.12     .05       0  141.47     .07       0
Bank Sta=93.12,141.47
Exp/Cntr=0.3,0.1

Type RM Length L Ch R = 1 ,37064   ,417.11,395.49,387.7
BEGIN DESCRIPTION:
36986.16
END DESCRIPTION:
XS GIS Cut Line= 5
  893020.0082613  811321.7815996  892982.5080713  811342.0940745
  892932.5088421  811349.9064861   892877.820937  811374.9066128
  892801.2586891   811406.156259
#Sta/Elev= 21
       0 1730.54   17.37 1715.86   45.81 1700.89   93.25  1690.5   96.52  1689.8
   97.41 1689.34   98.57 1689.29  106.36 1689.46  110.87 1689.37  131.07 1689.35
  135.15 1689.08  142.24 1689.34  148.88 1689.45  159.53 1689.63  166.29 1690.27
  168.93 1690.34  189.66  1696.2  202.85 1701.41  210.06 1706.11  228.81 1719.79
  236.08 1725.69
#Mann= 3 , 0 , 0
       0    .085       0   93.25     .05       0  148.88    .075       0
Bank Sta=93.25,148.88
Exp/Cntr=0.3,0.1

Type RM Length L Ch R = 1 ,36669   ,438.35,416.44,379.58
BEGIN DESCRIPTION:
36590.67
END DESCRIPTION:
XS GIS Cut Line= 6
  892823.1330318  810956.1560272  892770.0080187  810982.7190459
   892709.070594  811020.2192359  892690.3210111   811035.844059
  892648.1331693  811053.0317741  892571.5709214  811103.0310033
#Sta/Elev= 28
       0 1760.81    9.72 1750.06   38.31 1722.04   61.86 1697.02   90.151688.737
   94.34 1687.51  100.91 1686.24  102.13 1686.22  109.48 1686.35  124.57 1686.26
   125.4 1686.33  131.09 1687.43  157.88 1692.44  163.45 1693.37  183.42 1695.53
  200.73 1697.28   215.9 1697.53   229.6 1697.36  235.58 1697.38   240.4 1698.23
  246.48 1699.03   251.6 1700.48  256.76 1701.65  285.08 1717.31  288.56 1718.66
  290.66 1720.51   292.1 1721.33  292.49 1721.48
#Mann= 3 , 0 , 0
       0     .09       0   90.15     .05       0  131.09     .07       0
Bank Sta=90.15,131.09
Exp/Cntr=0.3,0.1

Type RM Length L Ch R = 1 ,36252   ,465.34,461.54,448.76
BEGIN DESCRIPTION:
36174.23
END DESCRIPTION:
XS GIS Cut Line= 6
  892482.5086103  810667.0937268  892443.4455283  810704.5939168
  892418.4454016  810737.4064551  892396.5710589  810762.4065818
  892373.1338242  810784.2819486  892313.7582673  810853.0317849
#Sta/Elev= 24
       0 1731.07    1.96 1729.86   11.86 1721.87   33.39 1705.18   49.49 1694.62
   55.27 1690.99   71.61    1688   84.33 1685.87   95.52 1683.99   102.6 1683.91
   107.5 1683.98  119.27 1683.85  125.11 1683.43  130.861684.503  137.83 1685.79
   138.6 1685.99  138.85 1685.98  152.07 1690.04  160.85 1693.28  168.01 1695.68
  175.06 1697.75  202.66 1701.56  215.54 1704.63  251.52  1719.8
#Mann= 3 , 0 , 0
       0     .09       0   84.33     .05       0  130.86    .075       0
Bank Sta=84.33,130.86
Exp/Cntr=0.3,0.1

Type RM Length L Ch R = 1 ,35791   ,383.7,411.92,445.94
BEGIN DESCRIPTION:
35712.68
END DESCRIPTION:
XS GIS Cut Line= 6
  892090.3210434  810406.1563129  892048.1332016  810467.0937376
     892002.8206  810524.9064025  891976.2586055  810568.6561121
  891957.5079984   810590.531479  891904.3829853  810645.2193841
#Sta/Elev= 27
       0 1736.35   31.04 1710.58   48.31 1698.36   65.03 1686.19   82.19 1682.54
   88.211681.352   95.16 1679.98  100.21 1680.18   107.2 1680.59  131.84 1680.62
  145.96 1681.78  157.28 1683.98  163.31 1685.26  169.51 1686.88  175.71  1688.8
  180.02 1689.77  189.48 1692.41  211.52 1691.82  225.53 1691.59  244.83    1691
  245.72 1691.14  246.74 1691.42  264.72 1698.07  272.89 1703.37     291 1716.61
  301.31 1724.44  303.82 1726.26
#Mann= 3 , 0 , 0
       0     .09       0   88.21     .05       0  131.84    .075       0
Bank Sta=88.21,131.84
Exp/Cntr=0.3,0.1

Type RM Length L Ch R = 1 ,35379   ,400.98,440.35,438.42
BEGIN DESCRIPTION:
35300.76
END DESCRIPTION:
XS GIS Cut Line= 6
  891810.6330223  810174.9066774  891752.8203574  810215.5316272
  891716.8830594  810246.7812735  891682.5086533  810262.4060966
  891662.1961784  810268.6566403  891602.8206215  810296.7815268
#Sta/Elev= 24
       0    1723    3.53 1720.55   21.45 1707.79   55.46 1692.43   65.92 1689.13
   87.11 1685.04  106.221681.113  117.53 1678.79  139.15 1678.96  146.13 1678.83
  152.14 1679.05  156.04 1679.28   163.3  1679.7  173.49 1681.23   181.6 1683.44
  187.17 1684.75  189.64 1686.53  195.68 1692.61  200.85  1698.9  217.69 1713.98
   222.5  1718.4  227.38 1725.18  234.58 1733.26  243.01 1742.52
#Mann= 3 , 0 , 0
       0     .09       0  106.22     .05       0  156.04     .07       0
Bank Sta=106.22,156.04
Exp/Cntr=0.3,0.1

Type RM Length L Ch R = 1 ,34938   ,445.3,422.44,420.31
BEGIN DESCRIPTION:
34860.41
END DESCRIPTION:
XS GIS Cut Line= 6
  891679.3828694  809821.7811683  891645.0084633  809832.7193638
  891573.1338673  809834.2812317  891532.5078933  809851.4689468
  891509.0706586  809863.9690101  891474.6962526  809879.5938332
#Sta/Elev= 20
       0 1721.32   25.73  1700.3   34.28 1693.95   49.79 1686.58   51.24 1685.97
    76.7 1677.08   80.74 1675.64    85.9 1675.59  100.91 1676.01     124 1676.03
  131.261676.132  136.83 1676.21  145.08 1678.12   148.3 1679.16  156.01 1680.67
  158.07    1681  173.55 1685.23  197.42 1699.17  209.68 1705.49  216.42 1709.45
#Mann= 3 , 0 , 0
       0     .09       0    76.7     .05       0  131.26     .07       0
Bank Sta=76.7,131.26
Exp/Cntr=0.3,0.1

Type RM Length L Ch R = 1 ,34516   ,246.31,244.29,265.04
BEGIN DESCRIPTION:
34437.97
END DESCRIPTION:
XS GIS Cut Line= 6
  891468.4457088  809423.3440818  891407.5082841  809446.7813165
  891379.3833976  809462.4061397  891348.1337514  809481.1567468
  891310.6335614  809499.9063297  891243.4455929  809529.5941081
#Sta/Elev= 26
       0 1716.05       6 1712.29   61.791675.498   64.66 1673.61   74.99 1673.43
   82.49 1673.46   93.66 1674.41   102.2 1675.12  107.29 1676.08  108.83 1676.03
  111.42 1676.12  117.85 1676.73  136.62 1679.95  147.73 1683.32  152.96 1684.15
  160.55 1684.77  166.78 1684.86   177.1 1685.31  179.96 1685.77  187.54 1688.83
  202.54 1695.04  208.44 1697.78   222.6 1704.99  226.76 1706.72  236.86 1713.28
  249.29 1719.97
#Mann= 3 , 0 , 0
       0    .085       0   61.79     .05       0   93.66    .075       0
Bank Sta=61.79,93.66
Exp/Cntr=0.3,0.1

Type RM Length L Ch R = 1 ,34272   ,142.23,182.8,197.15
BEGIN DESCRIPTION:
34193.67
END DESCRIPTION:
XS GIS Cut Line= 6
  891387.1958092  809206.1563775  891295.0087382  809226.4688524
  891263.7580678  809248.3442193  891234.0713135  809259.2813906
  891198.1329913  809263.9690424  891149.6956299  809259.2813906
#Sta/Elev= 29
       0 1715.29   10.81 1712.58   23.21 1708.05   50.87 1696.81   82.08 1684.21
   82.15 1684.17   94.45 1679.41  105.82 1674.87  112.281673.744  116.32 1673.04
  117.28 1672.88  121.57 1671.92  126.04 1671.94  130.61 1672.37  133.65 1672.37
  136.72 1672.48  146.01 1673.19  155.56 1672.96   156.1 1672.97  157.06 1673.16
  164.24 1674.77   168.5  1675.7   173.4 1677.63  176.79 1679.03  200.48 1699.75
  203.43 1702.25     239 1737.49  239.23 1737.72  249.14 1747.37
#Mann= 3 , 0 , 0
       0    .085       0  112.28     .05       0  146.01    .075       0
Bank Sta=112.28,146.01
Exp/Cntr=0.3,0.1
