HEC-RAS study lds_big_laurel_crk.prj: lds_big_laurel_crk

--- lds_big_laurel_crk.g20 (geometry) --- (continued)

Type RM Length L Ch R = 1 ,34089   ,204.6,138.23,104.27
BEGIN DESCRIPTION:
34010.88
END DESCRIPTION:
XS GIS Cut Line= 6
  891359.0709227  809092.0939396  891271.5704794   809068.656705
  891243.4455929   809068.656705  891207.5082949   809068.656705
    891187.19582   809068.656705  891145.0079782  809096.7815914
#Sta/Elev= 23
       0 1706.38     .65 1706.08    4.09 1704.99   17.18  1701.7   39.69 1693.37
   63.58 1684.08   90.58 1674.04   96.74 1671.63  107.14 1671.41  117.74 1671.41
  119.61 1671.27  131.65  1670.8  134.31 1671.04  135.31 1671.03  145.37 1671.69
   151.1 1672.01  169.06 1690.17  181.61 1700.04  190.41 1708.76  200.16  1717.5
  210.59 1724.72  215.06 1727.41  225.66  1736.1
#Mann= 3 , 0 , 0
       0    .085       0  107.14     .05       0  145.37    .075       0
Bank Sta=107.14,145.37
Exp/Cntr=0.3,0.1

Type RM Length L Ch R = 1 ,33951   ,248.23,243.94,210.36
BEGIN DESCRIPTION:
33872.64
END DESCRIPTION:
XS GIS Cut Line= 6
  891280.9457829  808867.0938237  891249.6961366  808887.4062986
  891232.5084215  808912.4064253  891218.4454662  808929.5941404
  891199.6958833  808943.6560716  891145.0079782  808992.0944571
#Sta/Elev= 26
       0 1719.87   37.27 1692.53   39.03 1691.29   45.57 1685.18   63.73 1674.34
   66.22 1673.04   67.61 1672.71   73.92 1671.28   79.31 1670.17   86.03 1669.78
   89.75 1669.64   89.82 1669.64   94.04 1669.55   97.59 1669.98  104.65 1670.21
  113.25 1671.19  113.74 1671.24  119.48 1671.86  122.72 1672.14  123.16 1672.17
  123.87  1672.3  134.12 1672.74  137.53 1672.34  144.27 1675.81  156.48 1682.13
  186.31 1698.35
#Mann= 3 , 0 , 0
       0    .085       0   73.92     .05       0  113.74    .075       0
Bank Sta=73.92,113.74
Exp/Cntr=0.3,0.1

Type RM Length L Ch R = 1 ,33707   ,495.2,450.82,360.05
BEGIN DESCRIPTION:
33628.71
END DESCRIPTION:
XS GIS Cut Line= 5
   891055.945667  808740.5313225  891023.1331288  808787.4068161
  891002.8206539  808817.0935704  890984.0710709  808854.5937604
   890963.758596  808940.5313118
#Sta/Elev= 27
       0    1702   15.26 1687.37   34.731669.268   36.04 1668.05   41.51 1667.74
   45.71 1667.51   49.89 1667.59   52.36  1667.5   65.69 1666.92   66.17  1666.9
   74.311668.095   86.67 1669.91    88.8 1670.07   93.19 1670.18   93.82  1670.2
  118.68 1670.85  128.63 1669.71  129.72 1669.63   130.5 1669.79   133.8 1670.65
  135.12 1671.02  136.23  1671.3  145.28 1673.87  152.78 1675.36  168.85 1680.49
  187.43 1691.19  223.42 1712.65
#Mann= 3 , 0 , 0
       0    .095       0   34.73     .05       0   74.31    .075       0
Bank Sta=34.73,74.31
Exp/Cntr=0.3,0.1

Type RM Length L Ch R = 1 ,33256   ,460,456.78,453.17
BEGIN DESCRIPTION:
33177.89
END DESCRIPTION:
XS GIS Cut Line= 6
  890560.6338578  808643.6565998  890570.0081371  808693.6568532
  890582.5082005  808743.6560823  890609.0712191  808799.9068794
  890615.3207387  808823.3441141  890623.1331503  808893.6568424
#Sta/Elev= 30
       0 1706.53    6.88 1700.74   17.91 1692.25   32.38 1680.35   37.59 1676.75
   40.44 1674.99   50.39 1669.95   60.48 1669.44   72.29 1668.61   87.93 1665.83
   91.22 1664.98   92.22 1665.05  101.83 1664.72  107.44 1664.66  114.91  1664.9
  121.161666.041  135.28 1668.91  144.66 1671.32  146.84 1672.03   147.3  1672.1
  180.68 1675.61   186.6 1675.85  195.47 1676.08  200.97 1676.71  204.79 1677.03
  207.84 1679.01  228.74 1691.32     242  1693.7  255.38 1699.54  259.68 1701.62
#Mann= 3 , 0 , 0
       0     .09       0   87.93     .05       0  121.16    .075       0
Bank Sta=87.93,121.16
Exp/Cntr=0.3,0.1

Type RM Length L Ch R = 1 ,32799   ,451.44,430.79,411.12
BEGIN DESCRIPTION:
32721.11
END DESCRIPTION:
XS GIS Cut Line= 5
   890109.070734   808732.718911  890132.5079687  808832.7194177
  890159.0709873  808912.4064253  890180.9463542  808967.0943304
  890201.2588291  809009.2811481
#Sta/Elev= 30
       0 1710.23    8.48 1701.66   21.04 1690.01    27.7 1685.31      34 1680.22
   39.58 1675.92   51.53 1670.58   53.18 1670.05   55.23 1669.59   79.56  1666.8
   84.12 1666.36   96.63 1664.28  101.74 1663.52  115.47 1662.83  132.61 1662.55
  143.61  1662.6  148.791663.494  167.53 1666.93  181.15 1669.88  186.98 1670.79
  208.98 1672.11  213.71 1672.17  224.14 1672.72  226.78 1672.73  234.67  1676.7
   256.2 1687.84  263.57 1692.36  271.44 1698.23  287.75 1708.65  292.43 1711.49
#Mann= 3 , 0 , 0
       0    .085       0  101.74     .05       0  148.79    .075       0
Bank Sta=101.74,148.79
Exp/Cntr=0.3,0.1

Type RM Length L Ch R = 1 ,32368   ,207.14,145.01,37.89
BEGIN DESCRIPTION:
32290.32
END DESCRIPTION:
XS GIS Cut Line= 6
  889659.0705022  808851.4690006  889696.5706922  808903.0311218
  889713.7584073  808932.7189002  889748.1338375  809040.5318185
  889780.9453516  809096.7815914  889834.0703647  809170.2190795
#Sta/Elev= 30
       0 1696.87   10.69 1690.79   12.23 1689.35   16.31 1686.57   26.02 1680.86
   45.68 1668.83   58.41 1665.55    62.5 1664.74   92.68 1662.72  130.37 1660.46
  135.72 1660.98  138.47 1660.92  144.751662.857   148.1 1663.89  149.27 1664.15
  158.38 1667.55  166.83 1667.28  176.56 1667.98  207.55 1668.47  213.36  1668.3
  221.27 1668.47  233.14 1668.05  247.28 1667.82   273.4  1667.1  290.12 1666.94
  310.08 1668.83  345.32 1693.49   352.1 1697.79  354.39 1699.34  366.98 1706.86
#Mann= 3 , 0 , 0
       0     .08       0   92.68     .05       0  144.75     .07       0
Bank Sta=92.68,144.75
Exp/Cntr=0.3,0.1

Type RM Length L Ch R = 1 ,32223   ,253.97,262.35,238.99
BEGIN DESCRIPTION:
32145.31
END DESCRIPTION:
XS GIS Cut Line= 6
  889507.5078743  809026.4688632  889593.4454257    809048.34423
  889654.3828504  809062.4061612  889718.4460591  809093.6568316
  889757.5081169  809129.5941297  889802.8207185  809190.5315544
#Sta/Elev= 30
       0 1742.53    2.24 1740.68    9.35 1733.42   11.88 1730.51   29.61 1717.57
   51.48 1699.94   55.18  1698.1   59.88 1694.97   63.73    1691   68.36 1687.97
   73.22 1682.02    79.6 1678.37   91.761663.224   93.61 1660.92  142.93 1660.17
  148.81 1659.41  151.67    1661   158.3 1663.31  163.25  1666.2  166.83 1666.32
  175.29 1667.48   186.7 1667.84  214.14 1668.24  235.37 1668.03  268.18 1666.78
  290.77 1667.03  327.12  1689.8  338.69 1697.49  343.85 1700.67  351.51 1705.99
#Mann= 3 , 0 , 0
       0    .075       0   91.76     .05       0   158.3     .07       0
Bank Sta=91.76,158.3
Exp/Cntr=0.3,0.1

Type RM Length L Ch R = 1 ,31961   ,147.84,119.58,50.16
BEGIN DESCRIPTION:
31882.96
END DESCRIPTION:
XS GIS Cut Line= 6
  889413.7579114  809248.3442193  889465.3210567   809273.344346
  889548.1338483   809309.281644  889590.3206659  809326.4693591
  889620.0084443  809329.5941189  889685.6335208  809329.5941189
#Sta/Elev= 30
       0 1716.81    1.48 1715.51    3.53 1714.18   12.65 1704.03   21.86 1694.15
   24.94 1689.93   39.85 1673.67   46.47 1667.88    51.8 1661.64   79.72 1660.49
   84.81 1660.03   99.45 1658.71  114.99 1658.72  120.75 1658.86  124.57 1659.19
  129.45 1659.35  132.72 1659.99  144.43 1662.68     149 1663.31   177.3 1665.85
  186.67 1666.74  193.86 1667.56  196.81  1667.7   210.3 1669.21  223.56 1670.35
   235.8 1675.98  248.01 1680.52  256.89 1684.22  267.72 1692.72  288.61 1705.78
#Mann= 3 , 0 , 0
       0    .075       0   84.81     .05       0  129.45    .075       0
Bank Sta=84.81,129.45
Exp/Cntr=0.3,0.1

Type RM Length L Ch R = 1 ,31841   ,213.36,158.01,75.94
BEGIN DESCRIPTION:
31763.38
END DESCRIPTION:
XS GIS Cut Line= 6
  889391.8835686  809415.5316703  889429.3837587  809406.1563667
  889529.3832412  809404.5934747   889571.571083  809395.2191954
  889613.7579006  809379.5943722  889687.1953886  809379.5943722
#Sta/Elev= 27
       0 1710.93    8.85  1699.9   21.04 1686.92   24.15 1681.55   39.56 1661.22
   43.54 1660.12   51.19 1657.29   96.95 1657.49  105.44 1658.52  116.62  1660.5
  121.38 1661.19  130.39 1661.91  136.56 1662.29  160.99 1665.54   166.8 1666.17
  185.45 1667.31  198.65 1667.48  208.72  1667.5  214.61  1667.2  220.62 1668.02
  225.72 1668.44  231.76 1669.58  234.42 1670.44  257.57 1675.87  278.04 1689.48
  297.55  1699.8  300.32 1700.86
#Mann= 3 , 0 , 0
       0    .075       0   51.19     .05       0  105.44    .075       0
Bank Sta=51.19,105.44
Exp/Cntr=0.3,0.1

Type RM Length L Ch R = 1 ,31683   ,273.99,301.15,331.36
BEGIN DESCRIPTION:
31605.37
END DESCRIPTION:
XS GIS Cut Line= 6
  889502.8212467  809612.4068997  889524.6955894  809571.7819499
  889563.7586714  809509.2816332  889602.8207292  809468.6566834
  889666.8829137  809435.8441452   889699.695452  809417.0935381
#Sta/Elev= 29
       0 1703.07   32.28 1669.59   46.14 1658.23   46.81 1657.68   54.02  1657.4
    56.4 1657.21   58.59 1656.93   81.52 1657.12  115.18 1657.77  125.74 1658.88
  131.02 1659.09  135.99 1660.16  144.12 1661.67  147.97 1662.61  153.15 1663.71
  166.68 1664.43  180.17 1665.39  187.93 1665.69  195.53 1666.36  203.67 1666.88
  206.04 1667.12  212.61  1667.4  216.49 1668.08  222.44 1670.32   232.9 1674.98
  238.34 1676.84  255.24 1684.28  262.37 1687.23  285.97 1697.54
#Mann= 3 , 0 , 0
       0    .075       0   46.14     .05       0  115.18    .075       0
Bank Sta=46.14,115.18
Exp/Cntr=0.3,0.1

Type RM Length L Ch R = 1 ,31382   ,144.72,180.27,266.85
BEGIN DESCRIPTION:
31304.22
END DESCRIPTION:
XS GIS Cut Line= 6
  889677.8211093  809798.3439336  889735.6337742   809754.594224
  889796.5711989  809724.9064456  889857.5086236  809687.4062556
  889885.6335101  809668.6566726   889940.320391  809629.5935906
#Sta/Elev= 26
       0 1715.47   10.44  1706.3   51.21 1661.97   56.95 1655.25   64.59 1653.99
   69.08 1653.13   102.1 1654.01  116.481654.281  129.13 1654.53  136.47 1654.79
  138.27 1655.02  139.76 1654.98  145.87  1655.3  150.57 1655.29  166.16 1654.61
  193.96 1653.14  209.67 1656.82  219.56 1657.65  223.19 1658.71  234.99 1662.72
  249.29 1667.71  269.45 1675.89  274.35  1677.7   277.1 1678.63  298.83  1689.4
  312.84 1695.66
#Mann= 3 , 0 , 0
       0    .075       0   64.59     .05       0  116.48    .075       0
Bank Sta=64.59,116.48
Exp/Cntr=0.3,0.1

Type RM Length L Ch R = 1 ,31202   ,82.74,139.89,191.57
BEGIN DESCRIPTION:
31123.95
END DESCRIPTION:
XS GIS Cut Line= 6
  889695.0088244  809881.1567252  889763.7586606  809903.0310679
  889807.5083702  809907.7187197  889935.6337634  809910.8434795
   889979.383473  809924.9064348  890012.1960112  809938.9693901
#Sta/Elev= 30
       0 1702.94    2.13 1701.68    3.53  1700.7    9.82  1695.4   13.83 1693.63
   18.79 1689.36   42.49  1675.7   46.76 1673.48   53.23 1669.81   69.51 1661.81
   70.29 1661.61   71.33 1661.04   83.97 1656.23   90.47 1654.68   96.68 1653.78
  103.43  1652.4  106.73 1651.72  111.48 1651.04  154.931652.422  189.37 1653.25
   191.1 1653.56  210.49 1654.82  212.12 1654.84  224.47 1655.72  243.57 1659.61
  289.04 1679.29   302.4 1685.56  318.75 1694.15  321.13 1695.14  326.02 1698.08
#Mann= 3 , 0 , 0
       0    .075       0  103.43     .05       0  154.93    .075       0
Bank Sta=103.43,154.93
Exp/Cntr=0.3,0.1

Type RM Length L Ch R = 1 ,31062   ,131.76,194.36,225.58
BEGIN DESCRIPTION:
30984.06
END DESCRIPTION:
XS GIS Cut Line= 6
  889677.8211093  809932.7188464  889729.3832304  809981.1562077
  889759.0710089  810006.1563344  889795.0083069  810026.4688093
  889854.3838638  810067.0937591  889907.5078528  810110.8434687
#Sta/Elev= 30
       0 1689.64   16.81 1681.91   23.63 1678.45   44.91 1670.79   53.06  1667.1
   62.78 1664.68   65.13 1664.61   70.16 1663.97   73.33 1662.61   76.91 1660.56
   81.36 1658.75   83.93 1658.74   90.45 1659.23  100.48 1658.17  104.34 1657.61
  118.69 1652.23  125.13 1650.78  131.68 1650.34  205.25 1648.19  212.68 1650.06
  219.65 1652.18  233.97 1660.07   242.4  1666.8  243.74  1667.6  244.99 1668.53
  260.81 1681.65  262.91 1683.21  286.09 1703.39  290.59 1707.61   291.6 1708.45
#Mann= 3 , 0 , 0
       0    .075       0  131.68     .05       0  212.68    .075       0
Bank Sta=131.68,212.68
Exp/Cntr=0.3,0.1

Type RM Length L Ch R = 1 ,30868   ,199.72,213.41,233.78
BEGIN DESCRIPTION:
30789.71
END DESCRIPTION:
XS GIS Cut Line= 6
  889595.0083177  809990.5315113  889621.5713363  810057.7194798
  889641.8838112  810107.7187089  889654.3828504   810143.656007
  889674.6963495  810184.2819809  889704.3831037  810232.7193423
#Sta/Elev= 30
       0 1679.28   15.79 1674.03   32.66 1669.22   37.14 1668.65   40.53 1668.08
   52.58 1665.73   58.88 1664.86      65 1663.38   69.33 1662.45   81.63 1660.09
   86.97 1659.33   92.46 1658.87  100.14 1658.79  104.48 1657.66  106.67 1657.01
  112.37 1655.19   116.7 1653.59  122.59  1651.9  129.86 1650.01  141.111649.048
  165.36 1646.99  206.48 1647.58  207.89 1648.16  209.69 1648.61  212.17 1649.25
  222.28 1656.62  229.41 1667.83  242.78 1684.06  253.02 1695.75   266.5 1713.62
#Mann= 3 , 0 , 0
       0    .075       0  141.11     .05       0  209.69    .075       0
Bank Sta=141.11,209.69
Exp/Cntr=0.3,0.1

Type RM Length L Ch R = 1 ,30654   ,413.17,391.11,373.79
BEGIN DESCRIPTION:
30576.30
END DESCRIPTION:
XS GIS Cut Line= 5
   889404.383632   810013.968746  889424.6961069  810085.8443662
  889448.1333416  810160.8437221  889457.5086451   810218.656387
  889463.7581647  810295.2186348
#Sta/Elev= 30
       0 1670.08    1.87 1669.92   11.84 1669.42   27.05 1667.54   36.52 1666.07
      43 1665.19   52.69 1664.22   56.97 1663.59    75.6 1661.38   88.35 1659.43
   95.31 1658.65   103.4 1657.93  105.97 1657.91  122.83 1656.76  125.48 1656.37
  127.13 1655.85  131.71 1654.79  134.51 1653.58  139.54 1651.72     147 1648.69
  150.17 1647.52  153.27 1646.77  155.84 1646.08  160.83 1646.34  173.34 1645.73
  183.07 1644.65  211.83 1646.06  233.37  1647.1  269.25 1674.78  288.65 1694.75
#Mann= 3 , 0 , 0
       0    .075       0  153.27     .05       0  211.83    .075       0
Bank Sta=153.27,211.83
Exp/Cntr=0.3,0.1

Type RM Length L Ch R = 1 ,30263   ,264.48,194.73,162.57
BEGIN DESCRIPTION:
30185.19
END DESCRIPTION:
XS GIS Cut Line= 3
    888995.00835  810110.8434687   889066.882946  810237.4059699
  889116.8831994  810320.2187615
#Sta/Elev= 27
       0 1678.76    6.73 1671.89    8.29 1670.38   15.88  1664.4   19.63 1660.92
   29.33 1653.52      34    1652   35.69 1651.63   42.01 1652.04   51.48 1652.18
   63.26 1652.66   64.63 1652.45   69.13 1651.53   82.93  1649.9   95.58 1649.28
   96.48 1649.14  106.89 1646.58  110.75 1645.38   118.5 1643.33  121.47 1642.46
  181.41 1639.89  188.24 1639.87  190.631641.385  212.78 1655.43  224.18 1662.96
  232.05 1667.25  242.28 1673.28
#Mann= 3 , 0 , 0
       0    .075       0  121.47     .05       0  190.63    .075       0
#XS Ineff= 2 , 0
       0   63.26    1654               0
Permanent Ineff=
       F       F
Bank Sta=121.47,190.63
Exp/Cntr=0.3,0.1

Type RM Length L Ch R = 1 ,30068   ,181.28,104.82,82.01
BEGIN DESCRIPTION:
29990.46
END DESCRIPTION:
XS GIS Cut Line= 5
  888743.4462396   810254.593685  888871.5706086  810328.0311731
  888926.2585137  810365.5313631  888973.1329831  810390.5314898
  889049.6962551  810413.9687244
#Sta/Elev= 30
       0 1707.35   22.64 1682.51   30.71 1674.31   45.37 1659.83    49.7  1659.5
   64.95 1657.18   69.24 1655.94    93.8 1657.96   98.06 1656.85  104.24 1654.86
  111.27 1653.45  117.44 1652.47  134.86 1647.99  140.92 1644.96  148.53  1644.5
   152.1 1644.66  163.55 1644.27   169.2 1643.62  177.95 1641.47   179.8  1640.8
  218.68 1638.37  222.54 1637.99   232.7 1638.21  238.611639.979  265.33 1647.86
  282.71 1652.62  300.81 1657.93  321.06 1663.21  330.79 1664.94  347.18 1669.28
#Mann= 3 , 0 , 0
       0    .075       0   179.8     .05       0  238.61     .08       0
Bank Sta=179.8,238.61
Exp/Cntr=0.3,0.1

Type RM Length L Ch R = 1 ,29964   ,216.71,122.34,35.88
BEGIN DESCRIPTION:
29885.64
END DESCRIPTION:
XS GIS Cut Line= 6
  888709.0708094  810470.2184974  888874.6953684   810460.844218
  888898.1336272  810456.1565662  888940.3204448  810468.6566296
  888984.0711786  810468.6566296  889040.3209515  810438.9688511
#Sta/Elev= 30
       0 1695.68    2.43 1693.13   22.84  1677.9   27.63 1674.63   35.95 1669.31
   42.18 1663.26   46.64 1660.12    63.7 1652.19   68.82 1651.02   76.07 1648.51
   92.79 1646.59  102.25 1645.87  114.24  1644.7   128.6 1644.28  137.95  1643.7
  142.15 1642.89  157.27 1639.45  164.06 1637.76  176.04 1636.78   189.8 1636.48
  198.64 1636.04  206.38 1639.65  223.24 1645.95   233.8 1649.11  244.83 1652.18
  277.55 1659.76  294.63 1662.45  306.26 1664.72  318.17  1666.8  341.15 1668.89
#Mann= 3 , 0 , 0
       0     .07       0  157.27     .05       0  206.38     .08       0
Bank Sta=157.27,206.38
Exp/Cntr=0.3,0.1

Type RM Length L Ch R = 1 ,29841   ,279.46,166.84,150.48
BEGIN DESCRIPTION:
29763.30
END DESCRIPTION:
XS GIS Cut Line= 6
  888871.5706086  810654.5936635  888923.1337539  810582.7190674
  888959.0710519  810551.4694212  888968.4463555  810529.5940543
  888974.6958751  810501.4691678  889013.7579329  810463.9689778
#Sta/Elev= 27
       0 1684.34    2.69 1681.72    2.96 1681.34   15.05 1671.44   16.96 1669.97
   27.22 1661.24   33.22 1657.41   39.76 1653.42   52.66 1648.67   65.29 1646.28
   90.94 1645.19   96.66  1644.1  104.64 1642.24  109.33 1640.82  113.16 1639.94
  115.89 1638.54  117.93 1637.72  121.12 1637.44  131.01 1637.15  143.29 1635.29
  163.94 1635.12  165.991636.631  184.94  1650.6  201.75 1658.42   215.5 1660.83
  232.44  1661.1  242.85 1663.82
#Mann= 3 , 0 , 0
       0     .06       0  121.12     .05       0  165.99     .08       0
Bank Sta=121.12,165.99
Exp/Cntr=0.3,0.1

Type RM Length L Ch R = 1 ,29674   ,371.97,348.58,334.86
BEGIN DESCRIPTION:
29596.46
END DESCRIPTION:
XS GIS Cut Line= 6
  889163.7586929  810781.1561647  889138.7585663  810732.7188033
  889129.3832627  810681.1566821  889126.2585029  810545.2188774
  889127.8203707  810499.9062758  889115.3213316  810440.5317431
#Sta/Elev= 30
       0 1701.72   11.42  1690.8   22.02 1679.58   26.27 1675.64   32.66 1671.35
   36.46 1668.52   39.81 1665.76   47.44 1658.67   54.97 1651.37   62.32    1649
    64.5 1648.95   78.45 1647.03   98.84 1645.44  116.94 1644.55  158.07 1644.48
  168.34 1643.73  182.44 1641.92  193.76 1639.49  197.93 1638.18  204.121635.743
  206.02 1635.06  216.87 1634.07  229.12 1634.42   242.9 1636.45   258.2 1639.02
  268.74  1643.1   273.2 1644.39  309.85  1658.3  314.95 1659.69  348.92  1670.1
#Mann= 3 , 0 , 0
       0    .055       0  204.12     .05       0   242.9     .08       0
Bank Sta=204.12,242.9
Exp/Cntr=0.3,0.1

Type RM Length L Ch R = 1 ,29326   ,264.21,344.76,403.02
BEGIN DESCRIPTION:
29247.88
END DESCRIPTION:
XS GIS Cut Line= 6
  889518.4460698  810695.2186133   889476.258228  810603.0315423
  889473.1334683  810523.3435105  889466.8829245  810490.5309723
  889454.3828612  810445.2193949  889462.1962969  810415.5316164
#Sta/Elev= 30
       0 1666.85    4.15 1665.17    7.05 1663.55    14.1 1661.62   21.63 1658.64
   23.03  1657.8   32.16 1653.18   36.11 1651.66   40.12 1649.06   43.96 1648.18
   47.15 1646.84   55.17 1645.54   72.73 1643.06   82.57 1642.34   94.43 1641.73
  107.08 1641.79  112.97 1641.57  127.39  1640.6  136.76 1638.41  140.07 1637.24
  156.09  1634.2  163.58 1633.32  191.43 1633.76  211.63 1634.74  218.28 1637.48
  256.29 1657.95  261.54 1659.71  265.28 1661.13  276.21 1665.65  292.24 1674.89
#Mann= 3 , 0 , 0
       0    .055       0  156.09     .05       0  191.43     .08       0
Bank Sta=156.09,191.43
Exp/Cntr=0.3,0.1

Type RM Length L Ch R = 1 ,28981   ,375.32,386.35,395.38
BEGIN DESCRIPTION:
28903.12
END DESCRIPTION:
XS GIS Cut Line= 2
  889735.6337742  810713.9692204  889854.3838638  810540.5312256
#Sta/Elev= 25
       0 1667.07     3.2 1665.08    8.71 1662.09   14.41 1659.21   18.79 1657.74
   20.74 1657.03   39.08 1646.32   45.56 1642.49   48.01  1641.5   56.42 1639.08
   56.86 1638.96   57.53 1638.89   69.02 1638.62   73.14 1637.87    76.4  1637.1
   80.87  1635.2   90.25 1632.53   92.66 1631.97   94.29  1631.8  106.25 1631.52
  135.94 1630.82  161.13 1630.47  161.951631.063  193.08 1653.56   210.2 1665.27
#Mann= 3 , 0 , 0
       0    .065       0  106.25     .05       0  161.95     .09       0
Bank Sta=106.25,161.95
Exp/Cntr=0.3,0.1

Type RM Length L Ch R = 1 ,28595   ,298.01,310.18,327.69
BEGIN DESCRIPTION:
28516.77
END DESCRIPTION:
XS GIS Cut Line= 2
  890049.6962013  810913.9692096  890196.5711773  810742.0941068
#Sta/Elev= 26
       0 1663.54   11.53    1656   15.05 1653.81   21.85 1650.41   25.25 1648.87
   30.81 1645.76   36.07 1642.86   38.47 1641.59   47.93 1637.02   56.45 1636.28
   58.91 1636.36   59.94 1636.32   66.13 1635.31   70.59 1634.67   72.32 1634.46
   74.01 1634.09    87.4 1631.21   87.82 1631.15   93.47 1630.26  112.34 1629.31
  115.53 1629.16  168.87 1627.27  172.051627.818  173.98 1628.15  194.94 1638.12
  226.08 1653.93
#Mann= 3 , 0 , 0
       0    .065       0  112.34     .05       0  172.05    .085       0
Bank Sta=112.34,172.05
Exp/Cntr=0.3,0.1

Type RM Length L Ch R = 1 ,28285   ,190.32,254.18,293.79
BEGIN DESCRIPTION:
28206.59
END DESCRIPTION:
XS GIS Cut Line= 4
   890257.508602  811120.2187184  890343.4461534  811038.9688188
  890427.8208128  810971.7818745  890462.1962431  810951.4693996
#Sta/Elev= 28
       0 1673.23    5.59  1671.2   11.19 1669.76   11.54 1669.63    11.9 1669.44
   32.57  1658.4   35.37 1655.74   38.81 1652.84   44.43 1647.91   53.44 1644.57
   53.52 1644.56   63.83 1644.24   68.94 1644.04   74.62 1643.21   75.62  1642.5
   78.67 1641.34   89.15 1636.65   94.48 1633.86   97.87 1632.85  114.38  1625.6
   131.8 1625.45  132.73 1625.45  177.18 1625.17  180.291626.214  186.29 1628.23
   222.4 1642.51  226.12 1645.37  266.05 1675.72
#Mann= 3 , 0 , 0
       0     .07       0  114.38     .05       0  180.29    .085       0
Bank Sta=114.38,180.29
Exp/Cntr=0.3,0.1

Type RM Length L Ch R = 1 ,28030   ,274.27,320.45,345.76
BEGIN DESCRIPTION:
27952.41
END DESCRIPTION:
XS GIS Cut Line= 4
  890321.5707865  811263.9689347  890398.1330344  811251.4688714
  890451.2580475  811245.2193518  890566.8833774  811237.4069402
#Sta/Elev= 29
       0 1666.84    6.99 1664.12     8.8 1663.27   16.54 1660.22   22.97 1658.23
   32.21 1655.07   38.65  1652.1   41.69 1651.01   47.64 1648.61   53.99 1646.33
   63.28 1642.31   75.42 1637.21   83.03 1635.58   88.78  1635.3   93.33 1634.84
   96.64 1634.77  103.31 1631.92  111.95 1628.98  113.58  1628.5  118.71 1627.23
  119.95 1626.64  142.51 1625.75  180.84 1625.36  184.571627.049   193.8 1631.23
  208.59  1636.2  217.69 1642.65  243.45 1662.37  246.96 1664.91
#Mann= 3 , 0 , 0
       0    .065       0  119.95     .05       0  184.57    .085       0
Bank Sta=119.95,184.57
Exp/Cntr=0.3,0.1

Type RM Length L Ch R = 1 ,27710   ,171.24,229.37,266.72
BEGIN DESCRIPTION:
27631.96
END DESCRIPTION:
XS GIS Cut Line= 4
  890279.3829448  811503.0309818  890377.8205595  811542.0940638
  890487.1963697  811578.0313618  890568.4462693  811603.0314885
#Sta/Elev= 30
       0    1660    4.65 1657.59    7.46 1656.26   12.33 1654.19   19.32 1650.75
   20.72 1649.95   24.28 1648.19   31.92 1644.95   36.62 1643.36   44.39 1640.06
   47.26 1639.43   56.08 1636.91   59.03 1635.92   63.55 1634.99      72 1633.66
   84.52 1632.23   90.57 1631.12   97.56  1629.1  105.91 1626.09  108.28 1625.25
   178.8 1624.94  184.55 1625.81  195.49 1627.66  219.75 1632.16  221.46 1632.87
  237.85 1641.05  283.08 1667.05  296.09 1674.68  297.23 1675.54  306.04 1678.74
#Mann= 3 , 0 , 0
       0     .06       0  105.91     .05       0  184.55     .08       0
#Block Obstruct= 1 ,-1
       0    11.21675.326
Bank Sta=105.91,184.55
Exp/Cntr=0.3,0.1

Type RM Length L Ch R = 1 ,27481   ,94.59,186.13,226.85
BEGIN DESCRIPTION:
27402.60
END DESCRIPTION:
XS GIS Cut Line= 3
  890188.7587658  811628.0316152  890271.5705332  811715.5310343
   890388.758755  811838.9687757
#Sta/Elev= 30
       0 1659.95    6.22 1657.91   11.12 1655.86   18.34 1651.07   20.07 1650.14
   32.99 1641.89   37.48 1639.46   46.26  1635.4   48.63 1635.41    51.5 1634.88
   55.43 1634.74    64.1 1634.03   79.57 1633.66  116.67 1627.59  122.07 1625.92
  136.19 1625.09  156.01 1623.93  201.55 1623.55  206.08 1624.42  210.55 1625.03
  215.41  1625.4  217.24 1625.96  223.37 1627.17  230.17 1630.42  241.35 1637.36
  243.33 1638.82  247.64 1641.53  270.23 1661.03  286.49 1676.16  290.68 1680.42
#Mann= 3 , 0 , 0
       0     .07       0  136.19     .05       0  206.08     .07       0
Bank Sta=136.19,206.08
Exp/Cntr=0.3,0.1

Type RM Length L Ch R = 1 ,27294   ,354.44,336.78,336.29
BEGIN DESCRIPTION:
27216.47
END DESCRIPTION:
XS GIS Cut Line= 3
  890134.0708607   811667.093673  890126.2584491  811795.2190662
   890146.570924  811895.2185487
#Sta/Elev= 24
       0 1651.13    3.94 1651.31    4.35 1651.26   16.05 1643.51    20.9 1640.89
   32.56 1634.42   33.23  1634.3    41.5 1633.54   50.36 1632.19   64.57  1626.6
   68.88 1624.34   78.66  1620.4   85.98 1620.16   89.54 1619.64   141.8 1619.27
  148.15 1620.43  154.45 1619.33  176.53 1625.96  176.98 1626.18     183  1633.4
   203.4 1657.15  206.21 1660.32  214.66 1666.91  230.41 1684.36
#Mann= 3 , 0 , 0
       0     .07       0   85.98     .05       0  148.15     .07       0
Bank Sta=85.98,148.15
Exp/Cntr=0.3,0.1

Type RM Length L Ch R = 1 ,26958   ,303.41,274.77,270.32
BEGIN DESCRIPTION:
26879.69
END DESCRIPTION:
XS GIS Cut Line= 3
    889773.13294   811667.093673  889785.6330033   811743.656945
    889810.63313  811903.0319844
#Sta/Elev= 26
       0 1656.29    9.97 1650.29   12.69 1648.77   14.02 1647.95   16.14 1646.19
   29.78 1635.87   31.73 1634.26   37.74 1628.85   48.71 1625.68   53.09 1624.69
   70.81 1622.33   74.57 1620.58   80.371617.478   82.46 1616.36  141.15 1616.33
  143.47 1616.78  152.26 1617.75  160.22 1619.53  167.41 1620.57  176.54  1621.7
  202.37 1631.52  205.84 1633.88  213.71 1637.28  223.19 1642.38  232.67 1647.88
   238.9 1651.77
#Mann= 3 , 0 , 0
       0    .085       0   80.37     .05       0  143.47     .07       0
Bank Sta=80.37,143.47
Exp/Cntr=0.5,0.3

Type RM Length L Ch R = 1 ,26683   ,83.76,99.86,77.95
BEGIN DESCRIPTION:
26604.92
END DESCRIPTION:
XS GIS Cut Line= 6
  889484.0706396  811631.1563749  889466.8829245  811695.2185594
  889487.1953994  811745.2188128  889513.7584181  811792.0943064
  889535.6337849  811882.7184853  889560.6328874  811934.2816307
#Sta/Elev= 30
       0 1664.82    4.21  1663.3   27.78 1657.42   35.19 1654.85    59.5 1639.55
    78.3 1631.88   84.78 1630.48  105.04  1629.6     113 1629.67  121.98 1628.63
  127.17 1627.69     133  1626.3  149.47 1618.84  152.92 1617.86  154.88 1617.18
  160.79 1617.07  197.53 1614.91  221.25 1615.08  223.71 1615.35  231.29 1617.51
  237.61 1619.56  243.35 1620.94   261.9 1623.64  265.91  1623.9   272.7 1625.16
  286.69 1630.25  304.03 1639.09  318.14  1647.4  321.52 1650.02  324.72 1651.15
#Mann= 4 ,-1 , 0
       0     .08       0   84.78     .06       0  152.92     .04       0
  231.29    .075       0
Bank Sta=152.92,231.29
Exp/Cntr=0.5,0.3

Type RM Length L Ch R = 3 ,26642   ,,,
BEGIN DESCRIPTION:
26569  FBSTR_1287  No Photo/Pier Data
END DESCRIPTION:
Bridge Culvert--1,0,-1,-1, 0
Deck Dist Width WeirC Skew NumUp NumDn MinLoCord MaxHiCord MaxSubmerge Is_Ogee
15,42,2.6,0, 5, 5, , , 0.95, 0, 0,0,,
     113   128.5     205   281.5     286
 1629.67 1629.91 1629.91 1629.91  1629.9
         1627.91 1627.91 1627.91
   63.29   123.5     200   276.5   339.5
 1629.57 1629.91 1629.91 1629.91  1629.9
         1627.91 1627.91 1627.91
Pier Skew, UpSta & Num, DnSta & Num=  ,179.5, 2 ,174.5, 2 , 0 , 0 , 0 ,,
       2       2
    1613    1628
       2       2
    1613    1628
Pier Skew, UpSta & Num, DnSta & Num=  ,230.5, 2 ,225.5, 2 , 0 , 0 , 0 ,,
       2       2
    1613    1628
       2       2
    1613    1628
BR Coef=-1 , 0 , 0 ,, 0 ,,,0.8,0,,0,
WSPro=,,,, 1 ,,,, 0 ,,,, 0 ,,,,-1 ,-1 ,-1 , 0 , 0 , 0 , 0 , 0
BR U #Sta/Elev= 61
       0 1664.82    2.61 1663.82    4.21  1663.3    7.17 1662.56   14.03  1660.7
   20.03 1659.43    22.3 1658.91   23.61 1658.54   27.78 1657.42   35.19 1654.85
   41.09 1651.16   47.76 1647.08   55.48 1642.12    59.5 1639.55   60.45 1639.31
   62.28 1638.36   66.33 1636.74    78.3 1631.88   84.78 1630.48   85.13 1630.45
   85.42 1630.44   86.38  1630.4   95.71 1629.91  105.04  1629.6     113 1629.67
  118.32 1629.11   120.3 1628.82  121.98 1628.63  127.17 1627.69  132.15 1626.61
     133  1626.3  135.38  1625.3  143.62 1621.62  149.47 1618.84  152.92 1617.86
  154.88 1617.18  160.79 1617.07   172.6 1616.15  197.53 1614.91  202.36 1614.94
  217.76 1615.07  221.25 1615.08  223.71 1615.35  225.611615.891  231.29 1617.51
  237.61 1619.56  243.35 1620.94  246.93 1621.49  251.81 1622.15  256.77 1622.85
   261.9 1623.64  265.91  1623.9  267.41 1624.15   272.7 1625.16  278.21 1627.22
  286.69 1630.25  299.58 1637.01  304.03 1639.09  318.14  1647.4  321.52 1650.02
  324.72 1651.15
BR U #Mann= 3
       0    .065   172.6     .04  225.61    .065
BR D #Sta/Elev= 82
       0 1664.27    1.73 1663.65    7.85 1662.16   10.54 1661.41   15.77    1658
   22.89 1653.22   23.76 1652.63    24.2 1652.36   25.47 1651.22   33.07 1644.59
   41.09 1637.14   42.16  1636.2   50.66 1630.41   51.68 1629.59   52.27 1629.37
   54.95 1629.41   63.29 1629.57   68.81 1629.35   72.55 1629.23   86.09 1628.62
    87.8 1628.53   91.63 1628.34   98.93  1628.1  104.08 1627.71  107.52 1627.44
  112.26 1627.26  113.52 1627.19  115.28 1627.07  120.83 1625.65  128.91 1625.03
  129.11 1625.03   132.5 1623.62  143.461617.342  145.14 1616.38  149.21 1615.76
  151.71 1615.22  169.98 1615.36  194.17 1614.55  196.32 1614.47  202.42 1614.17
  212.42 1613.89  220.88 1613.68  220.97 1613.68  227.43 1614.02   233.6 1613.96
  236.63 1614.99  244.42  1617.4   248.4 1618.17   257.4 1621.44  266.44 1623.85
  275.51 1625.98  275.69    1626  279.96 1626.41  284.79 1626.95  287.28 1627.26
  294.15 1627.52  296.71 1627.61  300.05 1627.86  303.69 1628.11  308.27 1628.34
  314.12 1628.58  314.21 1628.59   314.5  1628.6  315.53 1628.67  323.95 1629.35
  327.01 1629.63  330.69 1629.54  335.14  1629.3  338.82 1629.78  340.72 1631.06
  344.01 1633.99  349.14 1639.45  354.22 1642.76  357.01 1644.94   363.1 1649.71
  368.24 1653.16  374.84 1657.18  375.85 1658.09  376.99 1658.94  379.85 1660.81
   390.8  1667.2  393.54 1669.29
BR D #Mann= 3
       0    .065  143.46     .04  236.63    .065
BC Design=,, 0 ,, 0 ,,,,,,

Type RM Length L Ch R = 1 ,26583   ,107.86,160.29,225.39
BEGIN DESCRIPTION:
26505.06
END DESCRIPTION:
XS GIS Cut Line= 6
  889407.5083918  811637.4069187  889391.8835686  811723.3444701
  889398.1330882  811763.9694199   889441.883822  811862.4060104
  889491.8830512  811923.3444593  889557.5081277  811965.5312769
#Sta/Elev= 30
       0 1664.27   10.54 1661.41    24.2 1652.36   42.16  1636.2   51.68 1629.59
   72.55 1629.23  115.28 1627.07  120.83 1625.65  129.11 1625.03   132.5 1623.62
  143.461617.342  145.14 1616.38  151.71 1615.22  169.98 1615.36  220.88 1613.68
   233.6 1613.96  236.63 1614.99   248.4 1618.17   257.4 1621.44  275.51 1625.98
  287.28 1627.26  327.01 1629.63  335.14  1629.3  338.82 1629.78  344.01 1633.99
  349.14 1639.45  354.22 1642.76   363.1 1649.71   390.8  1667.2  393.54 1669.29
#Mann= 4 ,-1 , 0
       0     .08       0   51.68     .05       0  143.46     .04       0
  236.63     .07       0
Bank Sta=143.46,236.63
Exp/Cntr=0.5,0.3

Type RM Length L Ch R = 1 ,26423   ,433.54,396.29,342.77
BEGIN DESCRIPTION:
26344.76
END DESCRIPTION:
XS GIS Cut Line= 6
  889304.3831253   811629.593483  889277.8211308  811720.2186861
  889251.2581121  811813.9686491  889240.3209408  811846.7811873
  889229.3837694  811881.1566175  889221.5713579   811910.844396
#Sta/Elev= 29
       0 1665.03    2.98 1662.83    9.09 1657.49   21.14 1645.01   23.36 1642.52
   32.49  1632.8   43.17 1628.55   44.66 1628.46   57.11 1628.38   70.78 1627.15
   74.19 1626.27   83.93 1623.45   94.44 1615.97   96.47 1614.58   98.68 1614.24
   101.2 1614.55  102.17 1613.27  137.28  1613.8  169.01 1613.68  171.06 1614.38
  178.31 1615.02   186.1 1616.21  188.74 1616.37  200.32 1615.43  213.36 1615.52
  238.37 1625.87  240.15 1626.78  281.17 1646.54  293.24 1652.85
#Mann= 3 , 0 , 0
       0     .08       0   94.44     .05       0  171.06    .075       0
Bank Sta=94.44,171.06
Exp/Cntr=0.3,0.1

Type RM Length L Ch R = 1 ,26026   ,431.28,443.95,450.99
BEGIN DESCRIPTION:
25948.48
END DESCRIPTION:
XS GIS Cut Line= 4
  888849.6962659  811713.9691665  888882.5088041   811834.281124
  888893.4459755  811879.5937256  888896.5707352  811960.8436252
#Sta/Elev= 23
       0 1642.98   16.94 1628.81   25.57 1623.88   31.36 1623.65   33.16 1623.49
   40.17  1622.9   43.93 1622.28   51.44 1617.84   59.131613.958   64.85 1611.07
   68.85 1611.23  104.17 1611.61  119.29    1612  124.71 1612.13   155.7 1612.96
  165.12  1615.1  171.31 1617.52  178.88 1620.66  181.22 1621.78  207.72 1638.38
  215.84 1643.44  244.46 1665.13  252.63 1671.31
#Mann= 3 , 0 , 0
       0     .09       0   59.13     .05       0  124.71    .075       0
Bank Sta=59.13,124.71
Exp/Cntr=0.3,0.1

Type RM Length L Ch R = 1 ,25582   ,376.69,409.02,432.49
BEGIN DESCRIPTION:
25504.53
END DESCRIPTION:
XS GIS Cut Line= 4
  888430.9456803  811792.0943064  888443.4457436  811882.7184853
   888455.945807  811998.3438152  888465.3211105  812043.6564168
#Sta/Elev= 23
       0 1661.11   12.43  1649.7   45.18 1620.25   48.31 1620.28   51.22 1620.35
   55.84  1620.4    58.7 1620.39   65.46 1620.23   73.61 1620.13   74.54 1619.95
    75.5 1619.49   87.79 1612.94   90.75 1612.33   91.48 1612.22   97.23 1611.34
  148.45 1609.88  162.06 1609.42  180.52 1610.72  191.45 1613.95  203.65 1616.39
  207.78 1618.97  251.73 1646.71  254.05 1648.23
#Mann= 3 , 0 , 0
       0     .09       0   97.23     .05       0  180.52    .075       0
Bank Sta=97.23,180.52
Exp/Cntr=0.3,0.1

Type RM Length L Ch R = 1 ,25173   ,429.82,420.51,414.72
BEGIN DESCRIPTION:
25095.50
END DESCRIPTION:
XS GIS Cut Line= 3
  888076.2583034  811773.3436993  888043.4457652  811890.5319211
  888021.5703983  812032.7192454
#Sta/Elev= 26
       0 1659.69   25.04 1639.49   26.82 1637.98   29.03  1636.3   54.38 1619.81
   58.25 1618.73    70.7 1618.06   83.88 1616.36   97.11  1613.1  104.13 1611.54
  109.71 1610.36  113.01 1609.76  117.38 1609.16  119.36  1608.7  122.23  1607.3
  123.65 1607.03  179.46 1607.02  182.83 1607.03  186.59 1607.97  189.17 1608.59
  214.24 1613.87  219.44 1615.81  230.81  1620.3  241.72  1624.4  251.53 1627.45
  265.56 1634.31
#Mann= 3 , 0 , 0
       0    .085       0  119.36     .05       0  186.59    .075       0
Bank Sta=119.36,186.59
Exp/Cntr=0.3,0.1

Type RM Length L Ch R = 1 ,24753   ,452.4,444.3,433.74
BEGIN DESCRIPTION:
24675.00
END DESCRIPTION:
XS GIS Cut Line= 4
  887651.2581983   811704.593863  887637.1962671  811762.4065279
    887618.44566  811888.9690291  887612.1961405  811996.7819474
#Sta/Elev= 29
       0 1670.15   10.89 1659.52    16.9  1653.7   17.51    1653   18.02 1652.43
   55.74 1615.09    59.5 1614.41   62.83 1613.77    63.2 1613.81    64.8 1613.92
   74.12 1614.85   84.31 1614.53   85.55 1614.53   87.63 1614.11   98.39 1612.44
  104.38 1609.31  107.111608.371  111.91 1606.72  144.95  1606.1  187.32 1605.94
  187.44 1605.94  193.73 1605.95  198.221606.824  247.77 1616.47  250.28  1617.2
  289.87 1626.97  290.83 1627.18  294.28 1628.11  295.44 1628.44
#Mann= 3 , 0 , 0
       0    .095       0  107.11     .05       0  198.22    .075       0
Bank Sta=107.11,198.22
Exp/Cntr=0.3,0.1

Type RM Length L Ch R = 1 ,24309   ,186.11,215.13,253.85
BEGIN DESCRIPTION:
24230.70
END DESCRIPTION:
XS GIS Cut Line= 5
    887210.63327  811712.4062746  887187.1960353  811751.4693566
   887174.695972  811893.6566809  887182.5083835  811962.4065171
  887163.7588006  812012.4067705
#Sta/Elev= 26
       0 1647.95   14.14 1638.77   22.81 1633.45   35.61 1625.12   41.47 1621.62
   49.64  1615.8    55.6 1613.49   61.23  1613.3   68.32 1613.69   82.41  1609.4
   85.94 1608.39   91.77 1606.39   96.07 1605.68  103.38 1605.61  128.63 1605.77
  153.08 1606.57  188.98 1607.74   209.5 1611.86  222.41 1614.31  237.58 1616.14
  247.28 1617.06  261.57 1618.13  262.97 1618.91  293.17 1633.87  303.45  1639.2
  310.88 1643.18
#Mann= 3 , 0 , 0
       0    .085       0   85.94     .05       0  153.08     .08       0
Bank Sta=85.94,153.08
Exp/Cntr=0.3,0.1

Type RM Length L Ch R = 1 ,24094   ,136.6,206.59,296.31
BEGIN DESCRIPTION:
24015.57
END DESCRIPTION:
XS GIS Cut Line= 6
  887077.8212492  811626.4687232  887013.7580406  811696.7814514
  886984.0712863  811737.4064012  886979.3836345  811782.7190028
  886951.2587481  811876.4689658  886909.0709063  811942.0940422
#Sta/Elev= 30
       0 1657.23   21.36 1642.75   28.98  1638.3    59.6 1622.35   63.94 1619.69
    69.7 1619.62   82.09 1619.19    86.5 1618.77  108.73 1617.74  119.25 1616.83
  135.01 1614.38  145.44 1613.27  149.67 1613.33  163.78 1613.01  167.89 1612.61
  176.02 1610.91  180.65 1609.76  193.05 1606.51  197.741604.987  199.21 1604.51
  251.25 1604.36  276.21 1604.05  279.161604.816  291.86 1608.43   310.1 1612.33
  315.92 1613.94  319.68 1613.94  351.66 1630.86  358.29  1634.2  366.94 1639.85
#Mann= 3 , 0 , 0
       0     .08       0  197.74     .05       0  279.16    .075       0
Bank Sta=197.74,279.16
Exp/Cntr=0.3,0.1

Type RM Length L Ch R = 1 ,23887   ,188.12,235.01,229.63
BEGIN DESCRIPTION:
23808.98
END DESCRIPTION:
XS GIS Cut Line= 6
  886973.1330908  811553.0312351    886765.32069  811748.3435726
     886727.8205  811765.5312877  886688.7584421  811773.3436993
  886666.8830753  811773.3436993  886607.5085425  811759.2817681
#Sta/Elev= 30
       0 1660.58   15.83 1649.52   36.09 1634.99   62.44 1617.83   77.33 1616.73
      85 1617.74   95.47  1617.9  113.37 1617.24  161.32 1616.15  173.36 1614.26
  185.95 1612.85     203 1613.06  204.11 1612.46  210.78 1611.16  215.99  1607.9
  223.79 1606.02  234.08 1603.99  269.41  1605.1  280.12 1605.97  297.88 1606.16
  322.75 1608.38  343.44  1609.2  355.83 1610.93  375.25 1615.14  383.29 1619.62
  386.21 1620.33  388.18 1621.07  440.62 1643.96  443.52 1645.42   449.2 1649.04
#Mann= 3 , 0 , 0
       0     .08       0  223.79     .05       0  280.12    .075       0
#XS Ineff= 2 , 0
       0      85    1618               0
Permanent Ineff=
       F       F
#Block Obstruct= 1 ,-1
   90.97  143.171629.205
Bank Sta=223.79,280.12
Exp/Cntr=0.3,0.1

Type RM Length L Ch R = 1 ,23652   ,173.81,184.05,182.35
BEGIN DESCRIPTION:
23573.98
END DESCRIPTION:
XS GIS Cut Line= 6
  886832.5086584  811426.4687339  886780.9455131  811478.0318793
  886757.5082784  811496.7814622  886699.6956135  811526.4692406
  886620.0086059  811562.4065387   886502.820384  811596.7819689
#Sta/Elev= 30
       0 1662.63   13.24 1654.09   52.81 1623.39   62.66 1616.15   69.06 1614.95
   81.69 1613.57   98.44  1614.2  113.81 1614.48  121.62 1614.51  124.12 1614.68
  130.54  1614.8  136.14 1613.91  138.71 1613.78  142.96 1613.22   150.8 1612.77
  157.22 1612.18  167.48 1612.44  172.21 1612.72  176.83 1612.89   191.8 1606.28
  200.32 1603.49   202.7 1602.73  286.29 1602.84  291.41 1603.76  297.43 1604.84
  307.21 1606.19  313.66 1606.62  347.81 1633.55  357.41 1639.62  377.48 1652.91
#Mann= 3 , 0 , 0
       0     .08       0  200.32     .05       0  291.41     .07       0
Bank Sta=200.32,291.41
Exp/Cntr=0.3,0.1

Type RM Length L Ch R = 1 ,23468   ,385.2,419.37,424
BEGIN DESCRIPTION:
23389.93
END DESCRIPTION:
XS GIS Cut Line= 6
  886748.1329749  811303.0309925  886690.3213341  811337.4064228
   886637.196321  811360.8436575  886595.0084792  811378.0313726
  886476.2583896  811415.5315626  886452.8211549  811423.3439742
#Sta/Elev= 24
       0  1651.9   21.51 1639.32   24.65 1637.36   60.11 1615.97   78.21 1612.25
   80.55 1611.96   83.98 1612.09   92.77 1612.85  101.22 1612.77   104.2 1612.43
  121.77 1611.02  136.88 1611.94  141.21 1610.97  146.38 1609.95  156.25 1605.72
  167.311602.318  171.93 1600.92  252.34 1601.45   258.7 1602.49  260.45 1602.87
  288.34 1619.17   303.4 1629.88  316.84 1641.77  320.12 1644.77
#Mann= 3 , 0 , 0
       0     .08       0  167.31     .05       0   258.7     .07       0
Bank Sta=167.31,258.7
Exp/Cntr=0.3,0.1

Type RM Length L Ch R = 1 ,23048   ,348.09,415.62,461.5
BEGIN DESCRIPTION:
22970.56
END DESCRIPTION:
XS GIS Cut Line= 6
  886654.3830119  810965.5313308  886534.0710545  810970.2189825
  886459.0706745  810984.2819379  886416.8838568  810993.6562172
  886360.6330597  811012.4068243  886324.6957617  811012.4068243
#Sta/Elev= 30
       0 1641.64    7.06 1640.94   16.56 1639.07   17.47 1638.74   18.72 1637.94
   34.83 1626.09    46.4 1620.39   53.28 1617.18   56.47 1615.87   72.62 1612.12
   87.28  1610.6   94.09 1611.21  101.08 1611.24  104.38 1611.56  110.99 1611.81
  112.45 1611.59  120.33 1609.65  123.16 1609.69  132.83 1609.29  156.79 1608.85
  164.52 1608.52  171.92 1607.95  180.03 1606.12  194.73 1600.68  199.85 1598.63
  259.89  1597.8  261.231598.427   288.4 1611.14  304.93 1625.83  335.17 1649.91
#Mann= 3 , 0 , 0
       0    .065       0  199.85     .05       0  261.23    .075       0
Bank Sta=199.85,261.23
Exp/Cntr=0.3,0.1

Type RM Length L Ch R = 1 ,22633   ,337.07,366.68,352.95
BEGIN DESCRIPTION:
22554.93
END DESCRIPTION:
XS GIS Cut Line= 6
  886716.8833286  810640.5317323  886660.6335557  810634.2811886
   886560.633049  810603.0315423  886488.7584529  810582.7190674
  886445.0087433  810562.4065925    886395.00849  810557.7189407
#Sta/Elev= 30
       0  1637.2    4.15 1635.65   12.65 1633.17   15.89 1631.49   22.49 1628.57
   27.65 1625.47   42.63  1620.4    49.1 1618.68    54.4 1617.61   84.81 1614.73
   96.32 1612.53  103.39 1609.88  110.47 1610.34  145.31 1610.18   164.8 1609.58
  172.49 1607.99  180.58 1606.73  186.44 1604.59  194.52 1600.86  200.19 1599.65
  202.49 1598.47  207.91 1595.75  213.61 1596.71  234.31 1596.67  257.57  1599.2
  281.32 1601.74  308.16 1629.66  316.59 1636.68  323.98 1641.92  334.51 1648.36
#Mann= 3 , 0 , 0
       0     .07       0  202.49     .05       0  257.57    .075       0
#Block Obstruct= 2 ,-1
    48.8   80.611632.423  138.99  153.641620.472
Bank Sta=202.49,257.57
Exp/Cntr=0.3,0.1

Type RM Length L Ch R = 1 ,22266   ,255.49,315.34,359.57
BEGIN DESCRIPTION:
22188.26
END DESCRIPTION:
XS GIS Cut Line= 6
  886834.0705262  810356.1560595  886730.9462839  810284.2814635
  886663.7583155  810245.2194056  886616.8838461  810238.9688619
  886548.1329856  810238.9688619  886493.4461047  810213.9687352
#Sta/Elev= 30
       0 1633.63   18.18 1625.96   30.98 1621.24   42.54 1615.38   47.97  1613.4
   55.05 1612.34   74.41 1608.73   77.14 1607.55   83.67 1606.18   89.08  1606.8
  110.43 1607.74  116.11 1607.71  140.82 1608.84  155.79 1609.13  192.14 1607.13
  206.04 1607.02  210.21 1606.59  213.24  1604.3  218.45 1601.69  226.51 1597.13
  232.82 1594.72  235.12 1594.18  238.95 1594.44  247.45 1594.24  253.33 1594.59
  272.59 1596.95  319.46 1602.71  335.07  1603.9  362.59 1634.02  379.59 1653.27
#Mann= 3 , 0 , 0
       0     .06       0  226.51     .05       0  272.59    .075       0
Bank Sta=226.51,272.59
Exp/Cntr=0.3,0.1

Type RM Length L Ch R = 1 ,21951   ,179.06,261.91,293.33
BEGIN DESCRIPTION:
21872.91
END DESCRIPTION:
XS GIS Cut Line= 5
  886985.6331541  810138.9693794  886916.8833178  810104.5939491
  886798.1332282  810024.9069415  886760.6330382   809976.468556
  886680.9460306  809893.6567886
#Sta/Elev= 30
       0  1630.6    17.4 1622.42    28.6 1618.81   33.65 1615.87   39.14 1613.12
    43.2 1611.73   51.67 1607.58   65.05 1604.13   71.46 1603.67   97.63 1604.41
  108.71 1605.67  115.13 1606.08  131.58 1606.67     155 1607.92  186.58 1607.84
  207.43 1608.19  212.95 1607.83  217.66 1605.37  231.72 1598.91  237.56 1595.98
  241.15 1595.39   248.5 1596.34   255.91594.808  257.29 1592.61  321.71 1593.39
  322.461594.077  332.17 1603.13  336.06 1607.55  380.36 1648.78  396.06 1660.56
#Mann= 3 , 0 , 0
       0     .06       0   255.9     .05       0  322.46    .085       0
Bank Sta=255.9,322.46
Exp/Cntr=0.3,0.1

Type RM Length L Ch R = 1 ,21689   ,326.14,356.73,375.04
BEGIN DESCRIPTION:
21611.00
END DESCRIPTION:
XS GIS Cut Line= 6
  887079.3831171  810028.0317013  887049.6963628  809981.1562077
  887024.6962361  809937.4064981  886999.6961094  809865.5319021
  886987.1960461  809845.2194272  886949.6958561  809749.9065723
#Sta/Elev= 30
       0 1627.17    1.46 1626.56    6.71 1625.72    8.49 1625.25   17.22 1622.61
   32.04 1615.98   34.72 1614.72   38.92 1612.49   51.43 1607.39   56.66    1606
   59.16 1605.08   67.41 1603.62   72.68 1603.05   78.07 1602.76   89.48 1603.21
  103.34 1604.05  117.15 1604.21  136.28 1603.98  142.82 1603.67  153.49 1603.49
  159.77 1603.21  181.21 1594.07  185.75 1593.26  193.69  1592.7  203.47 1592.48
  247.61 1590.37  249.01 1590.49  253.881593.023  261.39 1596.93  308.25 1644.33
#Mann= 3 , 0 , 0
       0    .065       0  181.21     .05       0  253.88    .085       0
Bank Sta=181.21,253.88
Exp/Cntr=0.3,0.1

Type RM Length L Ch R = 1 ,21332   ,296.92,263.06,226.15
BEGIN DESCRIPTION:
21254.27
END DESCRIPTION:
XS GIS Cut Line= 4
  887363.7587899  809940.5312579  887354.3834863  809879.5938332
  887337.1957712   809754.594224  887324.6957079  809688.9691475
#Sta/Elev= 22
       0 1632.04   23.72 1619.67   38.81 1611.58   58.12 1601.68   74.77  1600.5
   82.48 1599.64   90.31 1598.08  111.25 1591.11  115.53 1589.78   124.3 1589.64
  132.18 1589.88  168.86 1590.13  175.57 1591.38  176.68 1591.22   180.1 1592.57
  187.83 1594.98   202.6 1599.22  203.38 1599.54  203.85 1599.64  204.56 1600.13
  236.67 1627.68  254.64 1643.39
#Mann= 3 , 0 , 0
       0    .075       0  111.25     .05       0  175.57    .095       0
Bank Sta=111.25,175.57
Exp/Cntr=0.3,0.1

Type RM Length L Ch R = 1 ,21069   ,218.2,159.01,98.68
BEGIN DESCRIPTION:
20991.21
END DESCRIPTION:
XS GIS Cut Line= 6
  887680.9459767  809829.5935799  887632.5086154  809779.5943507
  887604.3837289  809734.2817491   887584.071254  809703.0310787
  887543.4463042  809654.5937173  887493.4460508  809610.8440077
#Sta/Elev= 30
       0 1640.56     .99 1640.04   25.27 1625.37   39.99  1615.8   56.21 1606.66
   65.85 1601.86   68.97 1601.21   70.98 1600.66   85.62 1599.22   98.51 1597.18
  100.09 1596.68  113.891590.878  118.81 1588.81  119.36 1588.68  125.67 1588.15
  128.45 1588.06  174.63 1590.53  178.57 1590.71  180.13 1591.36   198.8 1597.02
  213.06 1599.56  218.94  1600.9  224.04 1605.47  226.63 1607.17  243.91 1621.57
  270.91 1643.54  271.72  1644.1  285.94 1655.27  286.45  1655.7  289.87 1659.03
#Mann= 3 , 0 , 0
       0    .075       0  113.89     .05       0  174.63     .08       0
Bank Sta=113.89,174.63
Exp/Cntr=0.3,0.1

Type RM Length L Ch R = 1 ,20910   ,431.77,398.1,378.54
BEGIN DESCRIPTION:
20832.20
END DESCRIPTION:
XS GIS Cut Line= 4
  887796.5713066  809615.5316595  887680.9459767  809578.0314695
  887593.4455334  809567.0942981  887523.1338293  809545.2189312
#Sta/Elev= 29
       0  1643.4   15.81 1629.84   21.85 1625.58   39.47 1612.65    52.7 1604.19
   63.09 1599.12   69.34 1598.96   72.58 1598.58   75.28 1598.42   77.92 1598.17
   83.72 1597.44   85.84 1596.97   87.68 1595.84   93.44 1591.61  102.87  1589.5
  105.42 1589.45  110.56 1588.53  116.33 1588.35  166.56 1588.88  205.69 1598.81
  209.13 1599.48  213.12 1600.37  217.17 1601.93  223.04 1605.38   236.3 1613.83
   251.2 1625.75  259.99 1632.02  265.01 1636.86  283.37 1652.62
#Mann= 3 , 0 , 0
       0    .075       0  105.42     .05       0  166.56    .075       0
Bank Sta=105.42,166.56
Exp/Cntr=0.3,0.1

Type RM Length L Ch R = 1 ,20512   ,268.14,261.72,252.84
BEGIN DESCRIPTION:
20434.10
END DESCRIPTION:
XS GIS Cut Line= 6
  887887.1954855  809173.3438393  887820.0085413   809179.594383
  887763.7587683  809184.2810106  887720.0080346  809185.8439026
  887663.7582616  809190.5315544  887605.9455967  809195.2192061
#Sta/Elev= 26
       0 1664.22    8.13 1659.01   23.07 1648.24   35.31 1636.49   51.21 1617.81
   67.95  1597.4   88.03 1596.96   92.41 1596.64  103.01 1595.09  105.24 1594.57
  115.62 1591.63  123.57 1588.92  125.64 1587.77  128.15 1587.88  183.77 1586.36
  187.081587.424   199.3 1591.35  210.09 1593.83  217.15 1593.79  221.13 1593.87
  251.79 1611.72  261.22    1617  266.07 1620.14  273.07 1625.45  279.58 1630.08
  282.15 1631.82
#Mann= 3 , 0 , 0
       0    .075       0  123.57     .05       0  187.08    .075       0
Bank Sta=123.57,187.08
Exp/Cntr=0.3,0.1

Type RM Length L Ch R = 1 ,20250   ,181.21,184.99,170.38
BEGIN DESCRIPTION:
20172.38
END DESCRIPTION:
XS GIS Cut Line= 5
  887859.0705991  808906.1569057  887729.3833381  808920.2188369
  887671.5706732  808931.1560082  887610.6332485  808940.5313118
  887563.7587791  808949.9066153
#Sta/Elev= 30
       0 1663.74    6.36  1659.4   22.66  1645.9   41.94 1622.13   62.48 1597.36
   63.22 1597.36   68.29 1595.18   76.39 1595.99  101.28 1596.72  109.78 1595.22
  116.24 1593.41  124.19 1590.54  125.92 1588.66  128.79 1587.96  130.45 1587.03
  133.56 1585.28  167.41 1585.42  177.41 1585.71  192.04 1585.39  195.57 1586.48
  198.35 1586.55  203.61 1588.51  215.21 1590.36  228.91 1593.11  235.01 1593.02
  246.72 1594.68  269.81 1607.39  277.66 1611.99  289.23 1619.61  298.74 1627.19
#Mann= 3 , 0 , 0
       0     .07       0  130.45     .05       0  195.57     .07       0
Bank Sta=130.45,195.57
Exp/Cntr=0.5,0.3

Type RM Length L Ch R = 1 ,20065   ,110.67,101.44,100.93
BEGIN DESCRIPTION:
19987.39
END DESCRIPTION:
XS GIS Cut Line= 6
  887857.5087313   808734.281803   887787.196003   808731.156019
  887646.5705465  808745.2189743   887584.071254   808768.656209
  887554.3834755  808787.4068161  887499.6955704  808838.9689373
#Sta/Elev= 30
       0 1671.37   23.48 1649.36   54.99 1610.64    66.6 1595.17  100.11 1596.73
   115.3 1596.46  116.29 1595.81  122.62 1593.76   129.3 1590.73  144.64 1586.89
   148.1 1586.01  211.71 1585.79  213.91 1585.81  217.69 1586.41  225.84 1587.87
  241.41 1593.17  248.92 1594.21  272.23 1598.42  286.03 1599.33  289.26 1600.01
  293.25 1601.58  300.36 1603.48  312.51 1610.28  322.18 1618.44  325.05 1619.67
  341.52 1621.67  361.82 1637.72  367.52 1641.64  370.59 1644.14  388.73 1654.71
#Mann= 3 , 0 , 0
       0     .07       0  144.64     .05       0  217.69    .065       0
#XS Ineff= 2 , 0
       0  135.45    1602  236.37       0    1602
Permanent Ineff=
       F       F
Bank Sta=144.64,217.69
Exp/Cntr=0.5,0.3
