HEC-RAS study lds_little_rock_crk.prj: Little Rock Creek Limited Detail Study

--- lds_little_rock_crk.g01 (geometry) --- (continued)

Type RM Length L Ch R = 3 ,33267   ,,,
BEGIN DESCRIPTION:
Little_Rock_Crk_96
Structure ID: Roan Mountain Road side street 6
Approximate Survey Structure
END DESCRIPTION:
Bridge Culvert--1,0,-1,-1, 0
Deck Dist Width WeirC Skew NumUp NumDn MinLoCord MaxHiCord MaxSubmerge Is_Ogee
24,15,3,0, 60, 60, , , , 0, 0.5,0.5,,
  4431.1  4433.7  4440.3  4457.4  4460.7  4476.8  4484.7  4493.6  4512.9  4544.4
  4571.6  4615.2  4626.5    4645  4654.3  4695.5  4711.5  4737.5  4794.5  4818.6
  4831.3    4839  4845.9  4896.7  4922.2    4946    4961    4967    4967    5033
    5033    5104  5106.6    5132    5148  5279.6    5373    5414    5470  5481.8
  5491.6  5501.4  5529.8  5542.8  5555.1    5566  5591.4  5604.9  5617.7  5640.5
    5651  5658.8  5669.6  5674.4    5678  5693.4  5726.4    5738  5749.7  5760.7
 3121.63 3120.69 3119.22 3114.63 3113.14 3109.52 3108.46 3106.59 3104.47 3099.44
 3095.86 3091.85 3090.35  3089.3 3089.16 3086.92 3085.64 3085.34 3085.36 3086.33
 3087.27 3086.63 3086.47 3087.16 3087.24 3086.92    3085  3084.5  3084.5  3084.5
  3084.5    3085 3086.05 3086.54 3087.17 3094.63 3098.25 3099.02 3098.65 3099.17
  3099.1 3100.42 3103.37 3105.17 3109.06 3111.07 3111.14 3111.57 3112.34 3114.41
 3116.14 3119.47 3122.92 3123.93 3126.09  3134.2 3151.22 3156.48 3162.37 3167.45
 3052.96 3052.96 3052.96 3052.96 3052.96 3052.96 3052.96 3052.96 3052.96 3052.96
 3052.96 3052.96 3052.96 3052.96 3052.96 3052.96 3052.96 3052.96 3052.96 3052.96
 3052.96 3052.96 3052.96 3052.96 3052.96 3052.96 3052.96 3052.96  3082.5  3082.5
 3052.96 3052.96 3052.96 3052.96 3052.96 3052.96 3052.96 3052.96 3052.96 3052.96
 3052.96 3052.96 3052.96 3052.96 3052.96 3052.96 3052.96 3052.96 3052.96 3052.96
 3052.96 3052.96 3052.96 3052.96 3052.96 3052.96 3052.96 3052.96 3052.96 3052.96
  4431.1  4433.7  4440.3  4457.4  4460.7  4476.8  4484.7  4493.6  4512.9  4532.7
  4544.4  4571.6  4615.2  4626.5    4645  4654.3  4695.5  4703.9  4711.5  4774.4
  4779.2  4798.3    4961    4967    4967    5033    5033    5104    5148  5170.1
  5182.3  5239.9  5279.6  5291.3  5310.4    5373    5414    5470  5481.8  5491.6
  5496.1  5501.4  5529.8  5542.8  5555.1    5566  5591.4  5604.9  5617.7  5640.5
    5651  5658.8  5669.6  5674.4    5678  5693.4  5726.4    5738  5749.7  5760.7
 3121.63 3120.69 3119.22 3114.63 3113.14 3109.52 3108.46 3106.59 3104.47 3101.45
 3099.44 3095.86 3091.85 3090.35  3089.3 3089.16 3086.92 3086.39 3085.64 3085.24
 3085.43 3085.45    3085  3084.5  3084.5  3084.5  3084.5    3085 3087.17  3088.6
 3089.01 3092.55 3094.63 3094.97 3095.97 3098.25 3099.02 3098.65 3099.17  3099.1
 3099.55 3100.42 3103.37 3105.17 3109.06 3111.07 3111.14 3111.57 3112.34 3114.41
 3116.14 3119.47 3122.92 3123.93 3126.09  3134.2 3151.22 3156.48 3162.37 3167.45
 3052.96 3052.96 3052.96 3052.96 3052.96 3052.96 3052.96 3052.96 3052.96 3052.96
 3052.96 3052.96 3052.96 3052.96 3052.96 3052.96 3052.96 3052.96 3052.96 3052.96
 3052.96 3052.96 3052.96 3052.96  3082.5  3082.5 3052.96 3052.96 3052.96 3052.96
 3052.96 3052.96 3052.96 3052.96 3052.96 3052.96 3052.96 3052.96 3052.96 3052.96
 3052.96 3052.96 3052.96 3052.96 3052.96 3052.96 3052.96 3052.96 3052.96 3052.96
 3052.96 3052.96 3052.96 3052.96 3052.96 3052.96 3052.96 3052.96 3052.96 3052.96
BR Coef= 1 , 1 , 0 ,1, 0 ,,,0.8,0,2,0,
WSPro=,,,, 1 ,,,, 0 ,,,, 0 ,,,,-1 ,-1 ,-1 , 0 , 0 , 0 , 0 , 0
BC Design=,, 0 ,, 0 ,,,,,,
BC HTab HWMax=3180.68

Type RM Length L Ch R = 1 ,33236   ,258,258,258
BEGIN DESCRIPTION:
Little_Rock_Crk_95
END DESCRIPTION:
XS GIS Cut Line= 2
      1075488.28       854981.91      1074481.34       855856.48
#Sta/Elev= 30
  4446.1 3119.22  4480.8 3107.01  4507.5 3100.44  4569.1 3092.25  4659.8 3083.83
  4750.6 3083.75  4902.2 3086.87  4958.9  3085.8  4967.5 3082.67    4992 3074.71
    4996  3072.3    5004  3072.3 5009.66 3074.22  5032.1 3080.65 5054.41 3082.91
 5107.84 3084.34  5127.3 3087.61  5171.7 3090.06  5354.2 3097.13  5450.5 3097.57
  5474.3 3098.76  5525.8 3103.59  5537.6 3105.51  5549.5 3109.11    5611 3112.24
  5633.5 3114.76    5645  3116.4  5680.8 3125.64  5754.2 3159.62  5779.8  3170.5
#Mann= 7 ,-1 , 0
  4446.1    .055       0  4659.8     .05       0  4967.5     .09       0
    4992    .052       0 5009.66     .09       0  5032.1     .05       0
  5680.8     .08       0
#XS Ineff= 3 ,-1
  4446.7    4891    3095    4891 4961.75    3087 5110.35 5120.95    3087
Permanent Ineff=
       T       F       F
#Block Obstruct= 1 ,-1
    4900    4952    3100
Bank Sta=4992,5009.66
Exp/Cntr=0.5,0.3

Type RM Length L Ch R = 1 ,32978   ,307,307,307
BEGIN DESCRIPTION:
little_rock_crk_a4
END DESCRIPTION:
XS GIS Cut Line= 3
      1075458.46       854802.03      1074933.37       855129.31
      1074300.39       855578.87
#Sta/Elev= 30
  4414.1 3112.17  4498.7 3098.21  4588.4 3088.82  4632.5 3085.36  4790.6 3078.55
  4888.7 3081.65  4952.5 3079.97  4972.8 3075.11  4981.4 3070.79  4983.9 3070.48
  4987.8 3068.43  5012.2 3068.43  5018.3 3069.93  5056.6 3082.55  5105.1 3082.04
  5292.7 3085.61  5416.5 3093.78  5490.9 3100.19  5522.3 3100.79  5543.4 3105.01
  5574.6 3107.26  5640.3 3110.08  5657.9 3112.59    5685 3118.21  5700.6 3118.93
  5714.1 3126.42  5735.9 3135.86  5745.9  3139.3  5775.7 3147.29  5809.2 3154.91
#Mann= 5 ,-1 , 0
  4414.1     .05       0  4952.5     .09       0  4983.9     .05       0
  5018.3     .09       0  5056.6     .05       0
Bank Sta=4983.9,5018.3
Exp/Cntr=0.3,0.1

Type RM Length L Ch R = 1 ,32671   ,632,632,632
BEGIN DESCRIPTION:
Little_Rock_Crk_94
END DESCRIPTION:
XS GIS Cut Line= 2
      1075164.07       854622.98      1074278.66       855202.41
#Sta/Elev= 30
  4636.2 3134.19  4710.9 3101.77  4724.9 3094.01  4766.1 3081.45  4791.1 3077.37
  4827.6 3074.32  4955.1 3076.24  4982.2  3066.5  4987.8 3063.44  5012.2 3063.44
 5018.35 3066.68  5031.5 3072.19  5036.7  3072.6  5138.6 3072.85  5180.1 3077.03
  5277.4 3075.82  5397.8 3077.38  5443.2 3082.21  5451.2 3081.61  5472.1 3085.27
  5486.9 3090.67    5508 3091.63  5517.2  3089.4  5532.9 3091.27  5564.6 3098.66
  5585.8 3105.26  5625.5 3119.93  5663.5 3136.47    5675 3140.37  5694.4 3144.25
#Mann= 5 ,-1 , 0
  4636.2     .09       0  4766.1     .05       0  4982.2     .05       0
 5018.35     .05       0  5532.9     .08       0
Bank Sta=4982.2,5018.35
Exp/Cntr=0.3,0.1

Type RM Length L Ch R = 1 ,32039   ,225,225,225
BEGIN DESCRIPTION:
Little_Rock_Crk_93
END DESCRIPTION:
XS GIS Cut Line= 2
      1074825.53       853950.24      1074178.83       854662.04
#Sta/Elev= 30
    4424 3107.35  4429.9 3106.03  4453.2  3106.4  4492.2 3103.05  4524.9 3096.52
  4535.2 3093.55  4580.6 3070.67  4592.8  3067.2  4600.2  3067.5  4638.5  3068.4
  4754.6 3068.45  4787.2 3066.66  4810.5 3059.01  4938.5 3060.49  4961.5  3060.9
  4972.1  3059.1  4987.8 3054.59  5012.2 3054.59  5017.2 3058.55  5029.2 3063.74
  5058.3 3064.75  5218.1 3067.84  5240.5 3077.14  5275.6 3076.59  5296.3 3077.55
  5309.6 3077.69  5321.9 3081.28  5338.4 3091.82  5346.6 3099.04  5385.7 3117.68
#Mann= 9 ,-1 , 0
    4424     .05       0  4524.9     .08       0  4600.2     .05       0
  4810.5    .035       0  4938.5     .09       0  4972.1     .05       0
  5017.2     .09       0  5058.3     .05       0  5296.3     .06       0
#XS Ineff= 2 , 0
       0  4634.4    3070  5110.2       0    3070
Permanent Ineff=
       F       F
Bank Sta=4972.1,5017.2
Exp/Cntr=0.5,0.3

Type RM Length L Ch R = 1 ,31814   ,60,60,60
BEGIN DESCRIPTION:
Little_Rock_Crk_92.75
END DESCRIPTION:
XS GIS Cut Line= 4
      1074862.32       853747.49      1074306.84       854193.44
      1074249.67        854249.6      1074032.02       854477.28
#Sta/Elev= 30
  4255.3 3097.67  4381.6 3086.41  4404.4 3082.89  4493.2 3077.83  4570.6 3068.86
  4665.8 3065.04  4784.8 3064.12    4799 3062.01  4836.8 3062.71  4872.6 3060.49
    4876 3058.85  4877.1 3060.26  4943.9 3061.27 4980.17 3060.64  4986.1  3058.9
 4988.63 3056.45    4990    3052    4996    3050  5022.6 3053.97  5031.2 3058.29
  5043.4 3060.93  5112.8 3064.56  5125.2 3070.93  5135.1  3072.9  5179.5 3073.44
  5217.9 3101.93  5240.8 3107.12  5251.5 3116.01  5280.1 3126.43  5362.7 3145.59
#Mann= 6 ,-1 , 0
  4255.3     .05       0  4836.8    .035       0  4943.9     .05       0
 4980.17     .05       0  5031.2     .06       0  5179.5     .07       0
#XS Ineff= 2 , 0
       0    4928    3068    5072       0    3068
Permanent Ineff=
       F       F
Bank Sta=4980.17,5031.2
Exp/Cntr=0.5,0.3

Type RM Length L Ch R = 3 ,31782   ,,,
BEGIN DESCRIPTION:
Little_Rock_Crk_92.5
Structure ID: Roan Mountain Road side street 5
Approximate Survey Structure
END DESCRIPTION:
Bridge Culvert--1,0,-1,-1, 0
Deck Dist Width WeirC Skew NumUp NumDn MinLoCord MaxHiCord MaxSubmerge Is_Ogee
24,14,3,0, 60, 60, , , , 0, 1,1,,
  4239.2  4241.6    4248  4255.1  4258.1  4287.9  4308.7  4314.2  4317.2  4334.7
  4358.8  4359.3  4360.4  4372.7    4401  4409.7  4418.4  4454.6  4459.6    4461
    4480  4508.9    4545  4568.5  4613.1    4644  4696.6  4798.7    4983    4983
    5017    5017  5080.4  5086.1  5092.4  5114.6  5123.5  5130.2  5142.2  5151.5
  5161.4  5168.3  5172.4  5182.8  5196.6  5204.8  5216.3  5220.3  5225.1  5231.8
  5238.6  5245.1  5258.7  5266.2  5278.1    5289  5299.9  5317.6  5344.4  5360.5
 3100.32 3099.62 3098.28 3097.24  3096.5 3092.76 3090.71 3089.44 3089.02 3088.05
 3085.97 3085.63 3085.76 3084.29 3081.59 3079.22 3080.37 3078.21 3077.44 3077.78
 3076.47 3073.62 3070.38 3068.69 3067.53 3066.32 3065.03    3065    3065    3065
    3065    3065 3065.03 3065.28 3066.06 3070.44 3071.63 3072.26 3072.71 3072.27
 3073.04 3075.58 3078.83 3088.98 3101.79 3106.97 3111.03 3111.81 3113.67 3115.33
 3118.07 3121.92  3126.5  3128.8 3130.48 3132.66 3135.17 3140.08 3145.71 3149.93
    3030    3030    3030    3030    3030    3030    3030    3030    3030    3030
    3030    3030    3030    3030    3030    3030    3030    3030    3030    3030
    3030    3030    3030    3030    3030    3030    3030    3030    3030    3064
    3064    3030    3030    3030    3030    3030    3030    3030    3030    3030
    3030    3030    3030    3030    3030    3030    3030    3030    3030    3030
    3030    3030    3030    3030    3030    3030    3030    3030    3030    3030
  4239.2  4241.6    4248  4255.1  4258.1  4287.9  4308.7  4314.2  4317.2  4334.7
  4358.8  4359.3  4360.4  4372.7    4401  4409.7  4418.4  4454.6  4459.6    4461
    4480  4508.9    4545  4568.5  4613.1    4644  4696.6  4798.7    4983    4983
    5017    5017  5080.4  5086.1  5092.4  5114.6  5123.5  5130.2  5142.2  5151.5
  5161.4  5168.3  5172.4  5182.8  5196.6  5204.8  5216.3  5220.3  5225.1  5231.8
  5238.6  5245.1  5258.7  5266.2  5278.1    5289  5299.9  5317.6  5344.4  5360.5
 3100.32 3099.62 3098.28 3097.24  3096.5 3092.76 3090.71 3089.44 3089.02 3088.05
 3085.97 3085.63 3085.76 3084.29 3081.59 3079.22 3080.37 3078.21 3077.44 3077.78
 3076.47 3073.62 3070.38 3068.69 3067.53 3066.32 3065.03    3065    3065    3065
    3065    3065 3065.03 3065.28 3066.06 3070.44 3071.63 3072.26 3072.71 3072.27
 3073.04 3075.58 3078.83 3088.98 3101.79 3106.97 3111.03 3111.81 3113.67 3115.33
 3118.07 3121.92  3126.5  3128.8 3130.48 3132.66 3135.17 3140.08 3145.71 3149.93
    3030    3030    3030    3030    3030    3030    3030    3030    3030    3030
    3030    3030    3030    3030    3030    3030    3030    3030    3030    3030
    3030    3030    3030    3030    3030    3030    3030    3030    3030    3064
    3064    3030    3030    3030    3030    3030    3030    3030    3030    3030
    3030    3030    3030    3030    3030    3030    3030    3030    3030    3030
    3030    3030    3030    3030    3030    3030    3030    3030    3030    3030
BR Coef= 1 , 1 , 0 ,1.25, 0 ,,,0.8,0,2,0,
WSPro=,,,, 1 ,,,, 0 ,,,, 0 ,,,,-1 ,-1 ,-1 , 0 , 0 , 0 , 0 , 0
BC Design=,, 0 ,, 0 ,,,,,,
BC HTab HWMax=3145.59

Type RM Length L Ch R = 1 ,31754   ,414,414,414
BEGIN DESCRIPTION:
Little_Rock_Crk_92.25
END DESCRIPTION:
XS GIS Cut Line= 4
      1074831.86       853693.19      1074253.68       854163.35
      1074200.52        854215.5      1073987.88       854427.13
#Sta/Elev= 30
  4227.1 3110.71    4259 3104.94  4270.6 3104.38  4296.9 3097.75  4319.6 3096.48
    4336 3092.24  4347.3 3091.34  4366.2 3086.15  4377.3 3084.58  4436.7 3076.86
  4523.3 3069.01  4561.7  3067.2    4973 3059.29    4985 3055.03    4990 3051.75
    4996 3049.75    5004 3049.75 5018.96 3054.29  5036.8 3059.33    5069 3062.86
  5085.6 3067.97  5103.1 3071.02  5137.1 3072.16  5156.3 3072.72    5187 3105.21
  5198.6 3111.03  5211.8  3113.6  5269.5 3130.45  5323.1 3142.82  5346.8 3150.11
#Mann= 4 ,-1 , 0
  4227.1     .05       0    4985     .05       0 5018.96     .09       0
  5137.1     .07       0
#XS Ineff= 2 , 0
       0    4958    3064    5042       0    3064
Permanent Ineff=
       F       F
Bank Sta=4985,5018.96
Exp/Cntr=0.5,0.3

Type RM Length L Ch R = 1 ,31340   ,567,567,567
BEGIN DESCRIPTION:
Little_Rock_Crk_92
END DESCRIPTION:
XS GIS Cut Line= 2
      1074241.76       853355.62      1073692.72       854290.95
#Sta/Elev= 30
  4263.9 3082.16  4291.1 3076.49  4350.4 3075.95  4396.4 3077.95    4416 3073.27
  4435.2 3064.74  4448.1 3062.38  4490.1 3057.21  4753.8 3053.33    4777  3045.6
  4785.3 3044.82  4795.5 3048.24  4908.6 3048.34  4977.7 3051.01 4984.37 3047.62
  4987.8 3044.08  5012.2 3044.08  5017.7 3048.29  5037.6 3055.08  5048.8 3061.67
    5061 3065.83  5088.5 3065.74  5096.2 3069.49    5112 3081.26  5130.5 3088.41
  5166.8 3105.67  5202.7 3116.24  5225.8 3124.83  5293.1 3142.28  5348.5 3164.61
#Mann= 5 ,-1 , 0
  4263.9     .09       0  4448.1     .05       0  4753.8     .06       0
 4984.37     .05       0  5017.7     .07       0
Bank Sta=4984.37,5017.7
Exp/Cntr=0.5,0.3

Type RM Length L Ch R = 1 ,30773   ,65,65,65
BEGIN DESCRIPTION:
Little_Rock_Crk_91
END DESCRIPTION:
XS GIS Cut Line= 4
      1073581.94       853029.65      1073321.47        853945.9
      1073367.05       854167.25      1073364.88       854167.25
#Sta/Elev= 30
  4322.1 3063.59  4390.7 3057.66  4550.1 3052.11    4646 3051.44  4675.4 3049.49
    4782 3048.59    4825 3045.84  4899.9    3045  4938.8 3045.65  4974.9 3048.63
  4985.1 3044.41    4987 3039.95    4992 3037.95    5008 3037.95    5013 3039.95
  5022.6 3041.18  5047.3 3049.08  5087.2 3048.27  5165.3 3054.61  5200.4 3054.44
  5228.1 3056.54  5267.3 3055.39  5284.8 3056.37  5313.4 3068.77  5349.4 3078.51
  5367.5 3091.75    5397 3097.05  5430.6 3106.14  5500.7 3114.39  5502.9 3113.53
#Mann= 4 ,-1 , 0
  4322.1     .05       0    4987     .05       0    5013     .05       0
  5200.4     .09       0
#XS Ineff= 2 , 0
       0    4953 3047.69    5047       0 3048.77
Permanent Ineff=
       F       F
Bank Sta=4987,5013
Exp/Cntr=0.5,0.3

Type RM Length L Ch R = 3 ,30742   ,,,
BEGIN DESCRIPTION:
Little_Rock_Crk_90
Structure ID: Roan Mountain Road side street 4
Approximate Survey Structure
END DESCRIPTION:
Bridge Culvert--1,0,-1,-1, 0
Deck Dist Width WeirC Skew NumUp NumDn MinLoCord MaxHiCord MaxSubmerge Is_Ogee
24.5,13,3,0, 60, 60, , , , 0, 1,1,,
  4322.6  4331.2    4344  4355.3    4366  4379.5  4414.8  4424.7  4426.3  4427.5
    4430  4439.8  4443.4  4509.1  4545.3  4606.9  4635.5  4759.3  4817.2  4818.7
  4832.4  4832.9  4858.4  4877.4  4906.1  4932.2  4960.9  4970.7  4977.5  4977.5
  5022.5  5022.5  5032.6  5035.7  5052.1  5062.3  5080.3  5112.1  5133.7  5153.7
  5169.2  5191.1  5216.2  5238.5    5248  5257.5  5311.3  5324.9  5330.5  5353.9
  5357.4  5369.6  5377.1  5381.5  5396.2  5408.7  5428.7  5430.1  5442.6    5474
 3062.89 3062.75 3061.96 3060.57 3060.56 3059.99 3057.54 3056.26 3055.08 3056.15
 3056.78 3055.82 3056.32 3053.98 3053.23 3050.64 3049.82 3047.02 3046.34 3045.35
 3044.37 3045.31 3044.87 3045.62 3045.67  3046.4 3048.44 3048.58    3048    3048
    3048    3048  3048.1 3049.13 3048.58 3047.84 3047.46 3048.38 3048.02 3048.86
 3051.25 3053.33 3053.79 3054.89 3054.08 3053.77 3054.38 3055.42  3056.2 3057.87
 3058.47 3063.57 3068.74 3072.59 3081.01 3086.38  3093.8 3094.17 3095.24 3099.36
 3017.95 3017.95 3017.95 3017.95 3017.95 3017.95 3017.95 3017.95 3017.95 3017.95
 3017.95 3017.95 3017.95 3017.95 3017.95 3017.95 3017.95 3017.95 3017.95 3017.95
 3017.95 3017.95 3017.95 3017.95 3017.95 3017.95 3017.95 3017.95 3017.95    3046
    3046 3017.95 3017.95 3017.95 3017.95 3017.95 3017.95 3017.95 3017.95 3017.95
 3017.95 3017.95 3017.95 3017.95 3017.95 3017.95 3017.95 3017.95 3017.95 3017.95
 3017.95 3017.95 3017.95 3017.95 3017.95 3017.95 3017.95 3017.95 3017.95 3017.95
  4322.6  4331.2    4344  4355.3    4366  4379.5  4414.8  4424.7  4426.3  4427.5
    4430  4439.8  4443.4  4509.1  4545.3  4606.9  4635.5  4759.3  4817.2  4818.7
  4832.4  4832.9  4858.4  4877.4  4906.1  4932.2  4960.9  4970.7  4977.5  4977.5
  5022.5  5022.5  5032.6  5035.7  5052.1  5062.3  5080.3  5112.1  5133.7  5153.7
  5169.2  5191.1  5216.2  5238.5    5248  5257.5  5311.3  5324.9  5330.5  5353.9
  5357.4  5369.6  5377.1  5381.5  5396.2  5408.7  5428.7  5430.1  5442.6    5474
 3062.89 3062.75 3061.96 3060.57 3060.56 3059.99 3057.54 3056.26 3055.08 3056.15
 3056.78 3055.82 3056.32 3053.98 3053.23 3050.64 3049.82 3047.02 3046.34 3045.35
 3044.37 3045.31 3044.87 3045.62 3045.67  3046.4 3048.44 3048.58    3048    3048
    3048    3048  3048.1 3049.13 3048.58 3047.84 3047.46 3048.38 3048.02 3048.86
 3051.25 3053.33 3053.79 3054.89 3054.08 3053.77 3054.38 3055.42  3056.2 3057.87
 3058.47 3063.57 3068.74 3072.59 3081.01 3086.38  3093.8 3094.17 3095.24 3099.36
 3017.95 3017.95 3017.95 3017.95 3017.95 3017.95 3017.95 3017.95 3017.95 3017.95
 3017.95 3017.95 3017.95 3017.95 3017.95 3017.95 3017.95 3017.95 3017.95 3017.95
 3017.95 3017.95 3017.95 3017.95 3017.95 3017.95 3017.95 3017.95 3017.95    3046
    3046 3017.95 3017.95 3017.95 3017.95 3017.95 3017.95 3017.95 3017.95 3017.95
 3017.95 3017.95 3017.95 3017.95 3017.95 3017.95 3017.95 3017.95 3017.95 3017.95
 3017.95 3017.95 3017.95 3017.95 3017.95 3017.95 3017.95 3017.95 3017.95 3017.95
BR Coef= 1 , 1 , 0 ,1.25, 0 ,,,0.8,0,2,0,
WSPro=,,,, 1 ,,,, 0 ,,,, 0 ,,,,-1 ,-1 ,-1 , 0 , 0 , 0 , 0 , 0
BC Design=,, 0 ,, 0 ,,,,,,
BC HTab HWMax=3114.39

Type RM Length L Ch R = 1 ,30708   ,545,545,545
BEGIN DESCRIPTION:
Little_Rock_Crk_89
END DESCRIPTION:
XS GIS Cut Line= 3
      1073514.44       853036.18      1073255.61       853936.74
      1073283.83       854114.69
#Sta/Elev= 30
  4344.6 3064.14  4361.8 3063.34  4370.6 3061.06  4372.1 3056.92    4377 3060.69
  4401.9  3055.9  4429.9 3056.91  4624.1 3049.58    4850 3043.89    4903 3045.47
  4906.2 3044.38  4908.2 3042.04  4910.6 3045.73  4957.1 3046.84  4979.5 3045.07
    4987  3039.7    4992  3037.7    5008  3037.7    5013  3039.7  5021.8 3039.31
  5051.2 3047.08  5142.4 3044.59  5183.3 3044.89  5193.7  3046.2  5218.7 3052.59
    5307 3052.95  5374.4 3056.53  5408.9 3061.45  5429.1 3070.25  5461.8  3066.5
#Mann= 4 ,-1 , 0
  4344.6     .05       0    4987     .05       0    5013     .05       0
  5429.1     .09       0
#XS Ineff= 3 ,-1
  4344.6    4950    3045    5050  5122.2    3045  5122.2  5461.8    3050
Permanent Ineff=
       F       F       F
Bank Sta=4987,5013
Exp/Cntr=0.5,0.3

Type RM Length L Ch R = 1 ,30163   ,482,482,482
BEGIN DESCRIPTION:
Little_Rock_Crk_88
END DESCRIPTION:
XS GIS Cut Line= 2
      1072792.61        853746.7       1073207.1       854406.42
#Sta/Elev= 30
    4868 3067.65  4883.1 3058.94  4935.4 3040.17  4945.1  3039.4  4964.7 3033.12
  4985.2 3032.64  4986.8 3031.05  5013.2 3031.05  5016.5 3032.77  5041.2  3036.3
  5052.9 3035.55  5055.7 3033.34  5059.4 3033.55    5064 3035.83    5079 3039.02
  5131.4 3041.26  5140.5 3042.83  5148.7    3046  5158.3 3051.86  5201.4 3052.54
  5238.3 3054.62  5305.5 3055.18  5330.9 3058.33  5407.8 3061.59  5468.9 3062.44
  5503.2 3067.89  5541.8  3073.2  5583.5 3082.21  5607.4 3084.59  5647.1  3092.3
#Mann= 4 ,-1 , 0
    4868     .09       0  4985.2     .05       0  5016.5     .05       0
  5503.2     .09       0
#XS Ineff= 2 , 0
       0                  5041.2       0    3040
Permanent Ineff=
       F       F
Bank Sta=4985.2,5016.5
Exp/Cntr=0.3,0.1

Type RM Length L Ch R = 1 ,29681   ,605,605,605
BEGIN DESCRIPTION:
Little_Rock_Crk_87
END DESCRIPTION:
XS GIS Cut Line= 2
      1072391.13       853698.95      1072352.07       854460.67
#Sta/Elev= 30
  4848.9 3058.68  4856.7 3056.08  4865.5 3051.69  4885.5 3044.65  4894.8 3042.24
  4901.1 3039.71  4935.1 3035.71  4965.9 3034.08  4981.2 3028.73 4984.86 3024.14
  4986.8 3021.39  5013.2 3021.39  5016.9 3021.92  5020.7 3023.42  5037.7 3032.95
  5057.4 3033.27  5079.8  3044.5  5082.3 3044.98  5133.8 3047.98  5184.4 3049.46
  5199.4 3050.71  5220.1 3052.86  5237.2  3053.1  5280.1 3057.06  5346.1 3060.74
  5498.9 3075.36  5536.3 3077.41  5548.4 3079.35  5568.5 3081.13  5611.6 3083.09
#Mann= 4 ,-1 , 0
  4848.9     .09       0 4984.86     .05       0  5020.7    .055       0
  5199.4     .05       0
Bank Sta=4984.86,5020.7
Exp/Cntr=0.3,0.1

Type RM Length L Ch R = 1 ,29076   ,378,378,378
BEGIN DESCRIPTION:
Little_Rock_Crk_86
END DESCRIPTION:
XS GIS Cut Line= 2
      1071787.83       853729.34      1071807.37       854445.48
#Sta/Elev= 30
  4854.7 3061.21  4858.3 3060.71  4878.6 3051.01  4915.2 3036.21  4933.3    3030
  4942.1  3028.4  4947.2 3026.83  4952.5 3023.98  4962.6 3017.68  4980.1 3008.14
  4986.8 3005.52  5013.2 3005.52 5017.15 3008.09  5033.1 3017.01  5068.8    3021
  5091.8 3028.49  5112.8 3036.23  5129.3 3040.52  5147.9 3043.53  5175.1 3046.74
  5210.4 3047.05  5216.3 3049.24  5219.4 3050.85  5221.2 3051.08    5227 3051.17
    5277  3055.9  5395.3 3068.81  5426.7 3071.47  5434.8 3072.74  5571.2    3084
#Mann= 3 , 0 , 0
  4854.7     .09       0  4980.1     .05       0 5017.15     .05       0
Bank Sta=4980.1,5017.15
Exp/Cntr=0.3,0.1

Type RM Length L Ch R = 1 ,28698   ,243,243,243
BEGIN DESCRIPTION:
little_rock_crk_a5
END DESCRIPTION:
XS GIS Cut Line= 3
      1071603.01       853654.74      1071419.58       853866.93
      1071466.34       854471.15
#Sta/Elev= 30
  4609.5 3047.72  4616.4 3044.93  4658.7 3036.62  4693.9 3028.86  4757.5  3018.9
  4780.7 3016.96  4803.3 3016.19  4849.4 3017.09  4874.6 3016.84  4901.3 3015.85
  4927.8 3011.86  4965.4 3011.32  4978.8 3010.17 4984.61 3004.28  4986.8 3002.03
  5013.2 3002.03  5028.4 3003.16  5038.3 3004.21    5052 3012.09  5072.7 3032.77
  5081.6 3040.97  5093.3 3041.05  5106.8 3040.14  5117.8 3044.75  5220.3 3050.26
    5302 3053.84  5389.4 3059.25  5415.3 3059.94  5456.7 3062.85    5496 3064.51
#Mann= 5 ,-1 , 0
  4609.5     .05       0  4965.4     .09       0 4984.61     .05       0
  5028.4     .09       0  5072.7     .05       0
Bank Sta=4984.61,5028.4
Exp/Cntr=0.5,0.3

Type RM Length L Ch R = 1 ,28455   ,80,80,80
BEGIN DESCRIPTION:
Little_Rock_Crk_85
END DESCRIPTION:
XS GIS Cut Line= 6
      1071495.71       853621.91       1071263.5       853860.63
      1071185.38       853977.82      1071128.95       854097.17
      1071165.85       854251.25      1071259.16       854518.18
#Sta/Elev= 30
  4534.7 3042.29  4594.4    3023  4611.2 3019.12  4639.3 3014.29  4659.3 3012.83
  4692.8 3013.05    4756  3011.2  4814.3 3006.22  4975.3 3002.86  4977.1 3002.74
  4987.2 2998.62    4996  2994.5    5004  2994.5  5008.5 2996.53  5011.4 2996.99
  5014.6 2998.74  5038.8 3017.83    5051 3019.57  5082.4 3019.45    5135 3021.98
  5140.6 3022.38  5175.3 3029.01  5196.2 3027.33  5204.9 3029.45  5213.7 3029.43
  5287.6 3034.15  5365.5 3036.55  5441.3 3043.13  5553.8 3049.74  5582.4 3052.04
#Mann= 3 ,-1 , 0
  4534.7     .05       0  4987.2     .05       0  5014.6     .05       0
#XS Ineff= 2 , 0
       0    4946    3004    5054       0 3006.24
Permanent Ineff=
       F       F
#Block Obstruct= 1 ,-1
    4786    4859    3025
Bank Sta=4987.2,5014.6
Exp/Cntr=0.5,0.3

Type RM Length L Ch R = 3 ,28410   ,,,
BEGIN DESCRIPTION:
Little_Rock_Crk_84
Structure ID: Roan Mountain Road side street 3
Approximate Survey Structure
END DESCRIPTION:
Bridge Culvert--1,0,-1,-1, 0
Deck Dist Width WeirC Skew NumUp NumDn MinLoCord MaxHiCord MaxSubmerge Is_Ogee
39,12,3,0, 60, 60, , , , 0, 1,1,,
  4552.9  4557.5  4568.6  4570.4  4582.7    4595    4616  4626.6  4637.6  4676.8
  4703.3    4727  4737.9  4759.6  4770.3  4781.3  4784.1  4797.1  4810.8  4824.7
    4856    4985    4985    5015    5015  5028.1  5031.7  5032.2  5043.7  5055.6
  5091.5  5130.8  5137.1  5139.9    5152  5159.4  5167.2  5189.1  5206.4  5217.9
  5227.7  5237.5  5248.4  5252.7  5258.7  5272.3  5301.3  5333.3    5345  5377.6
  5394.3  5407.8  5433.1  5440.1  5455.6  5487.3  5521.6  5558.2  5584.4  5600.6
 3033.21 3031.04 3026.97 3026.11 3021.46  3018.7 3015.34 3014.42 3013.79 3011.97
 3011.37 3011.13 3010.71  3008.6 3006.98 3006.54 3006.13 3005.29 3004.89 3004.13
    3004    3004    3004    3004    3004    3004 3004.51 3004.75 3005.76 3006.31
 3007.12 3008.32 3008.68 3009.78 3010.63 3010.09 3012.69 3018.51 3022.62 3026.91
 3025.79 3024.98 3025.82 3026.89  3027.7 3028.26 3030.08 3031.65 3031.93 3032.14
 3032.53 3033.25  3035.2 3036.25 3037.93 3040.64 3042.88 3044.71 3046.48 3047.88
  2974.5  2974.5  2974.5  2974.5  2974.5  2974.5  2974.5  2974.5  2974.5  2974.5
  2974.5  2974.5  2974.5  2974.5  2974.5  2974.5  2974.5  2974.5  2974.5  2974.5
  2974.5  2974.5    3002    3002  2974.5  2974.5  2974.5  2974.5  2974.5  2974.5
  2974.5  2974.5  2974.5  2974.5  2974.5  2974.5  2974.5  2974.5  2974.5  2974.5
  2974.5  2974.5  2974.5  2974.5  2974.5  2974.5  2974.5  2974.5  2974.5  2974.5
  2974.5  2974.5  2974.5  2974.5  2974.5  2974.5  2974.5  2974.5  2974.5  2974.5
  4552.9  4557.5  4568.6  4570.4  4582.7    4595    4616  4626.6  4637.6  4676.8
  4703.3    4727  4737.9  4759.6  4770.3  4781.3  4784.1  4797.1  4810.8  4824.7
    4856    4985    4985    5015    5015  5028.1  5031.7  5032.2  5043.7  5055.6
  5091.5  5130.8  5137.1  5139.9    5152  5159.4  5167.2  5189.1  5206.4  5217.9
  5227.7  5237.5  5248.4  5252.7  5258.7  5272.3  5301.3  5333.3    5345  5377.6
  5394.3  5407.8  5433.1  5440.1  5455.6  5487.3  5521.6  5558.2  5584.4  5600.6
 3033.21 3031.04 3026.97 3026.11 3021.46  3018.7 3015.34 3014.42 3013.79 3011.97
 3011.37 3011.13 3010.71  3008.6 3006.98 3006.54 3006.13 3005.29 3004.89 3004.13
    3004    3004    3004    3004    3004    3004 3004.51 3004.75 3005.76 3006.31
 3007.12 3008.32 3008.68 3009.78 3010.63 3010.09 3012.69 3018.51 3022.62 3026.91
 3025.79 3024.98 3025.82 3026.89  3027.7 3028.26 3030.08 3031.65 3031.93 3032.14
 3032.53 3033.25  3035.2 3036.25 3037.93 3040.64 3042.88 3044.71 3046.48 3047.88
  2974.5  2974.5  2974.5  2974.5  2974.5  2974.5  2974.5  2974.5  2974.5  2974.5
  2974.5  2974.5  2974.5  2974.5  2974.5  2974.5  2974.5  2974.5  2974.5  2974.5
  2974.5  2974.5    3002    3002  2974.5  2974.5  2974.5  2974.5  2974.5  2974.5
  2974.5  2974.5  2974.5  2974.5  2974.5  2974.5  2974.5  2974.5  2974.5  2974.5
  2974.5  2974.5  2974.5  2974.5  2974.5  2974.5  2974.5  2974.5  2974.5  2974.5
  2974.5  2974.5  2974.5  2974.5  2974.5  2974.5  2974.5  2974.5  2974.5  2974.5
BR Coef= 1 , 1 , 0 ,1.25, 0 ,,,0.8,0,2,0,
WSPro=,,,, 1 ,,,, 0 ,,,, 0 ,,,,-1 ,-1 ,-1 , 0 , 0 , 0 , 0 , 0
BC Design=,, 0 ,, 0 ,,,,,,
BC HTab HWMax=3052.04

Type RM Length L Ch R = 1 ,28375   ,661,661,661
BEGIN DESCRIPTION:
Little_Rock_Crk_83
END DESCRIPTION:
XS GIS Cut Line= 6
      1071401.55       853621.91      1071169.34       853860.63
      1071091.22       853977.82       1071034.8       854097.17
      1071071.69       854251.25        1071165.       854518.18
#Sta/Elev= 30
    4574 3021.16  4587.7 3017.03  4643.5 3015.81  4683.7  3013.2  4734.9 3011.35
  4793.8 3004.64  4968.2 3000.68  4982.9 2998.01    4996 2994.25    5004 2994.25
  5016.7 2997.69    5030 3003.15  5042.6 3000.98  5065.4 3002.01  5096.3 3001.64
  5147.5 2996.82  5173.6 2998.24  5179.9 2998.77  5184.6 3001.24  5194.3 3004.01
  5204.2 3005.15  5225.7 3015.78  5261.7 3022.94  5281.6  3023.1  5310.2 3026.67
  5356.7 3028.87  5441.1 3029.83  5513.4 3037.54  5571.1 3040.24  5621.8 3044.44
#Mann= 3 , 0 , 0
    4574     .05       0  4982.9     .05       0  5016.7     .05       0
#XS Ineff= 4 ,-1
    4574    4930    3008    4930    4956    3004    5044    5096    3004
    5096  5621.8    3008
Permanent Ineff=
       F       F       F       F
Bank Sta=4982.9,5016.7
Exp/Cntr=0.5,0.3

Type RM Length L Ch R = 1 ,27714   ,351,351,351
BEGIN DESCRIPTION:
Little_Rock_Crk_82
END DESCRIPTION:
XS GIS Cut Line= 2
      1070585.58       854164.45      1071217.09       854728.68
#Sta/Elev= 30
  4731.3 3059.02  4772.1 3040.65  4793.6 3032.62  4803.1 3027.23  4873.3 3002.09
  4902.1 2993.28  4916.2 2990.73  4952.5 2987.93  4958.9 2988.23  4979.9 2979.13
  4983.7 2978.85  4986.4 2977.61  5013.6 2977.61  5015.7 2979.55  5037.2  2981.6
  5043.9 2984.34  5065.6 2997.04  5091.8 3009.07  5112.4 3008.17  5119.8 3010.35
  5125.8 3014.84  5133.3 3018.27  5181.2 3023.09  5188.7 3024.59  5243.9 3027.51
  5373.5 3038.29  5394.9 3040.22  5401.3 3041.55  5444.8 3045.23  5578.1 3051.96
#Mann= 5 ,-1 , 0
  4731.3     .09       0  4803.1     .05       0  4983.7     .05       0
  5015.7     .09       0  5091.8     .05       0
Bank Sta=4983.7,5015.7
Exp/Cntr=0.3,0.1

Type RM Length L Ch R = 1 ,27363   ,380,380,380
BEGIN DESCRIPTION:
Little_Rock_Crk_81
END DESCRIPTION:
XS GIS Cut Line= 2
      1070420.65        854552.9      1071217.09       854932.68
#Sta/Elev= 30
  4708.9 3016.77  4743.1 3007.25  4790.9 2998.33  4802.1  2992.4  4833.5 2982.51
    4953 2978.38  4970.6 2979.73    4981 2977.55    4986  2975.7 4986.19  2974.2
  4986.4 2971.72  5013.6 2971.72  5017.6 2973.64  5048.5 2992.31  5075.8 2990.33
  5095.4 2993.39  5173.5 2997.57  5198.4 3000.43  5226.2 3007.77  5258.1 3012.32
  5401.4 3021.79  5419.2 3025.42  5440.8 3025.95  5460.5 3028.72  5473.6 3027.94
  5501.2 3033.01  5541.6 3036.92  5556.8 3036.54  5575.8  3040.6  5591.3 3041.01
#Mann= 3 , 0 , 0
  4708.9     .06       0 4986.19     .05       0  5017.6     .06       0
Bank Sta=4986.19,5017.6
Exp/Cntr=0.5,0.3

Type RM Length L Ch R = 1 ,26983   ,64,64,64
BEGIN DESCRIPTION:
Little_Rock_Crk_80
END DESCRIPTION:
XS GIS Cut Line= 2
      1070278.64       854676.95      1070736.11       855529.38
#Sta/Elev= 30
  4745.5 2998.95  4761.7 2993.32  4808.1  2984.5  4903.1 2975.46  4925.8 2974.24
    4964 2974.36  4977.5 2972.72    4986 2969.64    4995  2968.5    5005  2968.5
  5021.2  2971.6  5038.7 2973.78  5055.1 2974.67  5126.7 2975.73  5144.1 2977.08
  5151.9 2978.51  5166.4 2979.17  5195.2 2981.55  5221.7 2980.86  5334.4 2979.65
  5350.2 2981.04  5412.8  2987.2  5501.1  2992.9  5521.4 2995.33  5567.5 3002.78
  5645.6 3006.85  5653.8 3007.87  5683.6 3013.73  5705.1 3019.56    5713 3022.49
#Mann= 7 ,-1 , 0
  4745.5     .05       0  4977.5     .05       0  5021.2     .06       0
  5166.4    .035       0  5221.7    .025       0  5350.2    .035       0
  5501.1     .05       0
#XS Ineff= 2 , 0
       0    4950 2975.45    5050       0 2978.03
Permanent Ineff=
       F       F
Bank Sta=4977.5,5021.2
Exp/Cntr=0.5,0.3

Type RM Length L Ch R = 3 ,26950   ,,,
BEGIN DESCRIPTION:
Little_Rock_Crk_79
Structure ID: Roan Mountain Road side street 1
Approximate Survey Structure
END DESCRIPTION:
Bridge Culvert--1,0,-1,-1, 0
Deck Dist Width WeirC Skew NumUp NumDn MinLoCord MaxHiCord MaxSubmerge Is_Ogee
27,12,3,0, 60, 60, , , , 0, 1,1,,
  4763.3  4786.6  4805.5  4814.8  4847.2    4881  4969.6    4977    4977    5023
    5023  5041.4    5046  5047.9  5071.4  5080.3  5096.6  5109.4  5124.1  5153.8
    5160  5169.8  5173.8    5186  5204.3  5212.2  5231.9    5264  5296.7  5330.1
  5340.1  5344.1  5352.5  5363.1    5369  5381.2  5387.8  5392.1  5408.3  5414.1
    5424  5427.8    5435    5455  5470.6  5501.4  5527.6  5540.1  5565.7  5583.3
  5590.3  5602.8  5615.1  5625.8  5639.2  5651.5  5662.6  5683.1  5687.7  5730.3
 2990.72 2985.01  2982.6 2981.58 2979.29 2976.18 2977.65    2978    2978    2978
    2978 2977.75 2978.41 2978.34 2975.54 2975.54 2974.79 2974.76 2974.95 2976.72
  2976.4 2978.53  2978.6 2979.84 2980.96 2981.07 2980.49 2980.14 2980.14 2980.82
 2980.67 2980.96 2980.46 2980.87 2979.91 2980.12 2979.44 2979.82 2979.68 2982.06
 2983.28 2984.58  2985.6 2987.83 2989.22 2990.95 2993.73 2994.68  2997.7 2998.06
 2997.35 2995.46  2997.7 3000.02 3001.95 3006.07 3008.39 3013.31 3014.75  3025.5
  2948.5  2948.5  2948.5  2948.5  2948.5  2948.5  2948.5  2948.5    2976    2976
  2948.5  2948.5  2948.5  2948.5  2948.5  2948.5  2948.5  2948.5  2948.5  2948.5
  2948.5  2948.5  2948.5  2948.5  2948.5  2948.5  2948.5  2948.5  2948.5  2948.5
  2948.5  2948.5  2948.5  2948.5  2948.5  2948.5  2948.5  2948.5  2948.5  2948.5
  2948.5  2948.5  2948.5  2948.5  2948.5  2948.5  2948.5  2948.5  2948.5  2948.5
  2948.5  2948.5  2948.5  2948.5  2948.5  2948.5  2948.5  2948.5  2948.5  2948.5
  4763.3  4786.6  4805.5  4814.8  4847.2    4881  4969.6    4977    4977    5023
    5023  5041.4    5046  5047.9  5071.4  5080.3  5096.6  5109.4  5124.1  5153.8
    5160  5169.8  5173.8    5186  5204.3  5212.2  5231.9    5264  5296.7  5330.1
  5340.1  5344.1  5352.5  5363.1    5369  5381.2  5387.8  5392.1  5408.3  5414.1
    5424  5427.8    5435    5455  5470.6  5501.4  5527.6  5540.1  5565.7  5583.3
  5590.3  5602.8  5615.1  5625.8  5639.2  5651.5  5662.6  5683.1  5687.7  5730.3
 2990.72 2985.01  2982.6 2981.58 2979.29 2976.18 2977.65    2978    2978    2978
    2978 2977.75 2978.41 2978.34 2975.54 2975.54 2974.79 2974.76 2974.95 2976.72
  2976.4 2978.53  2978.6 2979.84 2980.96 2981.07 2980.49 2980.14 2980.14 2980.82
 2980.67 2980.96 2980.46 2980.87 2979.91 2980.12 2979.44 2979.82 2979.68 2982.06
 2983.28 2984.58  2985.6 2987.83 2989.22 2990.95 2993.73 2994.68  2997.7 2998.06
 2997.35 2995.46  2997.7 3000.02 3001.95 3006.07 3008.39 3013.31 3014.75  3025.5
  2948.5  2948.5  2948.5  2948.5  2948.5  2948.5  2948.5  2948.5    2976    2976
  2948.5  2948.5  2948.5  2948.5  2948.5  2948.5  2948.5  2948.5  2948.5  2948.5
  2948.5  2948.5  2948.5  2948.5  2948.5  2948.5  2948.5  2948.5  2948.5  2948.5
  2948.5  2948.5  2948.5  2948.5  2948.5  2948.5  2948.5  2948.5  2948.5  2948.5
  2948.5  2948.5  2948.5  2948.5  2948.5  2948.5  2948.5  2948.5  2948.5  2948.5
  2948.5  2948.5  2948.5  2948.5  2948.5  2948.5  2948.5  2948.5  2948.5  2948.5
BR Coef= 1 , 1 , 0 ,1.25, 0 ,,,0.8,0,2,0,
WSPro=,,,, 1 ,,,, 0 ,,,, 0 ,,,,-1 ,-1 ,-1 , 0 , 0 , 0 , 0 , 0
BC Design=,, 0 ,, 0 ,,,,,,
BC HTab HWMax=3022.49

Type RM Length L Ch R = 1 ,26919   ,317,317,317
BEGIN DESCRIPTION:
Little_Rock_Crk_78
END DESCRIPTION:
XS GIS Cut Line= 2
      1070225.69       854709.93      1070686.63       855571.91
#Sta/Elev= 30
  4760.7 2990.41  4791.4 2982.74  4813.7 2979.56  4909.3 2973.29  4961.7 2973.64
  4968.2 2973.02  4984.3 2974.46    4987 2970.75    4995 2968.25    5005 2968.25
    5013 2970.75  5038.8 2975.46  5070.8 2973.64  5113.2 2973.16  5142.2 2975.93
  5176.7 2977.42  5208.9 2980.51  5245.5 2980.48  5319.7 2981.26  5369.8  2982.4
  5383.5 2980.81  5446.4 2983.58  5482.9 2989.04  5622.4 2999.28    5650 3002.63
  5668.4 3006.19  5684.5 3009.52    5717 3019.89  5725.3 3021.55  5738.2 3022.44
#Mann= 6 ,-1 , 0
  4760.7     .05       0    4987     .05       0    5013    .055       0
  5176.7     .03       0  5245.5    .025       0  5319.7     .05       0
#XS Ineff= 2 , 0
       0    4952    2975    5048       0    2975
Permanent Ineff=
       F       F
Bank Sta=4987,5013
Exp/Cntr=0.5,0.3

Type RM Length L Ch R = 1 ,26602   ,365,365,365
BEGIN DESCRIPTION:
little_rock_crk_a6
END DESCRIPTION:
XS GIS Cut Line= 4
      1070031.33       854690.53      1070024.14       854974.66
      1070049.31       855060.97      1070081.68       855711.94
#Sta/Elev= 30
  4671.4 3005.99  4700.6 2997.02    4737 2983.83    4763 2976.09  4775.1 2973.02
  4808.8 2969.45  4848.3    2967  4880.8 2968.66  4906.4 2967.94    4940 2967.87
  4976.2 2969.38 4982.92 2965.65  4986.4 2963.39  5013.6 2963.39  5014.9 2965.55
  5048.4 2969.23  5085.8 2969.34  5137.1 2970.76    5160 2970.61  5178.4 2968.01
  5190.3 2969.98  5198.2 2972.96  5214.8 2974.01  5285.7 2973.14  5320.2 2973.84
    5549 2982.63  5602.9 2986.95  5640.3 2989.29  5661.3 2991.13  5697.3 2995.32
#Mann= 3 , 0 , 0
  4671.4     .06       0 4982.92     .05       0  5014.9     .06       0
Bank Sta=4982.92,5014.9
Exp/Cntr=0.3,0.1

Type RM Length L Ch R = 1 ,26237   ,727,727,727
BEGIN DESCRIPTION:
Little_Rock_Crk_77
END DESCRIPTION:
XS GIS Cut Line= 2
      1069819.52       854722.17      1069459.27       855338.49
#Sta/Elev= 30
    4815 2989.39  4853.3 2975.31  4872.4 2969.69    4889 2966.08    4932  2960.9
  4944.3 2960.76  4955.9    2959  4964.2 2959.32  4975.3 2956.51  4986.4 2954.88
  5013.6 2954.88 5014.22 2956.71  5014.6 2958.03  5025.5 2961.57  5056.1 2964.65
  5201.7 2967.81  5213.2 2965.18  5220.7  2963.7  5247.5 2966.53  5350.3 2969.48
  5359.3 2971.19  5370.3 2970.08  5377.3 2970.35  5383.5 2972.39  5411.3 2978.14
    5415 2981.53  5430.6 2987.77  5472.1 3006.65  5507.7 3017.52  5528.9 3023.09
#Mann= 6 ,-1 , 0
    4815     .09       0  4975.3     .05       0 5014.22     .05       0
  5213.2    .025       0  5350.3     .05       0  5383.5     .08       0
#XS Ineff= 2 , 0
       0                  5201.7       0 2967.81
Permanent Ineff=
       F       F
Bank Sta=4975.3,5014.22
Exp/Cntr=0.3,0.1

Type RM Length L Ch R = 1 ,25510   ,768,768,768
BEGIN DESCRIPTION:
Little_Rock_Crk_76
END DESCRIPTION:
XS GIS Cut Line= 2
      1069520.04       854055.94      1068884.19       854763.41
#Sta/Elev= 30
  4596.8  2985.1  4608.3  2982.3  4637.5 2979.51  4645.9 2975.82  4655.3 2975.25
  4666.9 2966.89  4670.2 2968.06  4671.9 2970.35  4684.5 2968.91  4877.6 2962.72
  4897.7 2960.91  4922.3 2949.59  4933.9 2948.05  4973.3 2949.08 4985.49  2947.2
  4986.4 2945.22  5013.6 2945.22 5015.53 2947.41  5018.8 2950.21  5072.6 2954.83
  5117.3 2955.99  5144.4 2954.48  5155.3 2958.49  5186.9 2976.21  5213.2 2976.65
  5302.2 2995.59  5344.1 3002.15  5475.9  3017.2  5508.1 3022.66    5548 3026.93
#Mann= 3 , 0 , 0
  4596.8     .08       0 4985.49     .05       0 5015.53     .05       0
Bank Sta=4985.49,5015.53
Exp/Cntr=0.3,0.1

Type RM Length L Ch R = 1 ,24742   ,403,403,403
BEGIN DESCRIPTION:
Little_Rock_Crk_75
END DESCRIPTION:
XS GIS Cut Line= 2
      1068712.75        853862.8      1068257.02       854468.27
#Sta/Elev= 30
    4783 3010.31  4798.6 3002.39  4813.3 2993.14  4826.5 2983.45  4835.3 2978.43
  4902.9 2944.77  4932.6 2936.09  4956.8 2931.41  4972.3 2930.06 4982.07 2927.01
  4985.9 2924.95  5014.1 2924.95  5028.7 2926.81  5049.8  2944.3    5062  2945.5
  5085.1 2952.87  5193.4 2956.44  5200.6 2960.33  5212.2 2963.63  5221.4 2965.67
  5241.1 2967.94  5250.2 2974.46    5305 2997.77  5337.7 3010.36  5359.3 3015.82
    5394 3021.66  5482.4 3032.51    5496 3035.09  5507.2 3035.31  5540.9 3039.51
#Mann= 4 ,-1 , 0
    4783     .09       0 4982.07     .05       0  5028.7     .05       0
  5250.2     .08       0
Bank Sta=4982.07,5028.7
Exp/Cntr=0.3,0.1

Type RM Length L Ch R = 1 ,24339   ,464,464,464
BEGIN DESCRIPTION:
little_rock_crk_a7
END DESCRIPTION:
XS GIS Cut Line= 2
      1068549.57       853503.69      1067977.72       854115.09
#Sta/Elev= 30
  4682.7 3054.97  4732.4 3037.83  4779.5  3015.4  4806.6 3000.92  4843.3 2985.74
  4848.6 2982.06  4873.3 2969.32  4885.1 2968.59  4920.6 2945.49  4951.8 2926.42
  4971.3  2916.1  4985.9 2912.41  5014.1 2912.41  5031.4 2917.96  5068.3 2921.15
  5084.7 2925.01  5100.9 2933.09  5141.1 2936.27  5154.8 2936.07  5170.4 2941.66
  5180.5  2952.3  5211.6 2981.27  5234.7 2990.33  5243.8 2992.34  5264.9 2993.99
    5289 2999.72  5375.9 3007.64    5441 3015.61    5463 3017.29  5519.8 3023.88
#Mann= 4 ,-1 , 0
  4682.7     .09       0  4971.3     .05       0  5031.4     .09       0
  5170.4     .06       0
Bank Sta=4971.3,5031.4
Exp/Cntr=0.5,0.3

Type RM Length L Ch R = 1 ,23875   ,232,232,232
BEGIN DESCRIPTION:
Little_Rock_Crk_74
END DESCRIPTION:
XS GIS Cut Line= 6
      1067826.14       852764.21      1067813.12       853068.03
      1067982.39       853460.82      1068038.81       853578.01
      1068078.81       853635.08      1067899.92        854007.7
#Sta/Elev= 30
3285.871 2962.083302.647 2955.123362.858  2944.63380.171    29393457.004 2935.27
 3458.69 2929.383462.215 2934.913482.668 2932.343498.831  2944.93518.825 2948.89
3559.042 2966.463588.612 2965.343600.256  2967.63657.862 2958.18 3696.93 2955.29
3726.118 2943.43 3783.57 2911.583808.773 2904.61 3811.07    29003822.562    2897
3837.883    28973849.373    29003854.965 2904.613879.172 2907.993911.269 2924.23
4060.418 2931.214143.074 2982.914171.571    29964199.839  3001.84316.123 3010.37
#Mann= 5 ,-1 , 0
3285.871     .09       03302.647     .05       03482.668     .09       0
3808.773     .05       03854.965     .06       0
#XS Ineff= 2 , 0
       03749.021    29283911.422       0    2928
Permanent Ineff=
       F       F
Bank Sta=3808.773,3854.965
Skew Angle= 40
Exp/Cntr=0.5,0.3

Type RM Length L Ch R = 3 ,23744   ,,,
BEGIN DESCRIPTION:
Little_Rock_Crk_73
Structure ID: Roan Mountain Road bridge
Approximate Survey Structure
END DESCRIPTION:
Bridge Culvert--1,0,-1,-1, 0
Deck Dist Width WeirC Skew NumUp NumDn MinLoCord MaxHiCord MaxSubmerge Is_Ogee
101,60,3,40, 60, 60, , , , 0, 1,1,,
3341.1033343.8613350.9853358.6453382.0863396.1813453.8653470.4873489.6383501.512
3522.1953523.7283535.6783538.3593542.0353544.8713546.1733546.3253547.398 3549.62
3562.1833578.1943728.5683752.6983757.4483757.4483902.9963902.9963909.0473920.232
3924.829  3931.83945.1293970.4084004.2684023.419 4066.244074.5144078.5754090.217
4105.6154121.931 4136.87 4149.284155.9444165.5964188.5014211.2524227.7224235.919
4244.1924257.6754259.8964266.4084275.5234292.6844311.6044346.0764364.2324386.907
 2947.27 2945.99 2942.05 2940.34  2938.3 2936.78 2934.58 2933.06 2930.01 2929.06
 2927.88 2927.55 2929.43 2930.49 2930.29 2928.36 2924.91 2919.09 2926.52 2929.76
 2929.67 2929.02 2929.06 2928.63    2928    2928    2928    2928 2928.31 2927.94
 2928.13 2927.62 2927.87 2927.75 2928.21 2928.79 2928.85 2930.37 2931.82 2937.89
 2947.37 2958.14 2968.48 2977.49 2981.82 2988.49 2990.53 2993.46 2996.96  2998.2
 2998.88  2999.1 2998.89 2997.52 2996.71 2997.42 2999.18 3001.41 3003.55 3007.16
    2877    2877    2877    2877    2877    2877    2877    2877    2877    2877
    2877    2877    2877    2877    2877    2877    2877    2877    2877    2877
    2877    2877    2877    2877    2877  2925.5  2925.5    2877    2877    2877
    2877    2877    2877    2877    2877    2877    2877    2877    2877    2877
    2877    2877    2877    2877    2877    2877    2877    2877    2877    2877
    2877    2877    2877    2877    2877    2877    2877    2877    2877    2877
3341.1033343.8613350.9853358.6453382.0863396.1813453.8653470.4873489.6383501.512
3522.1953523.7283535.6783538.3593542.0353544.8713546.1733546.3253547.398 3549.62
3562.1833578.1943728.5683752.6983757.4483757.4483902.9963902.9963909.0473920.232
3924.829  3931.83945.1293970.4084004.2684023.419 4066.244074.5144078.5754090.217
4105.6154121.931 4136.87 4149.284155.9444165.5964188.5014211.2524227.7224235.919
4244.1924257.6754259.8964266.4084275.5234292.6844311.6044346.0764364.2324386.907
 2947.27 2945.99 2942.05 2940.34  2938.3 2936.78 2934.58 2933.06 2930.01 2929.06
 2927.88 2927.55 2929.43 2930.49 2930.29 2928.36 2924.91 2919.09 2926.52 2929.76
 2929.67 2929.02 2929.06 2928.63    2928    2928    2928    2928 2928.31 2927.94
 2928.13 2927.62 2927.87 2927.75 2928.21 2928.79 2928.85 2930.37 2931.82 2937.89
 2947.37 2958.14 2968.48 2977.49 2981.82 2988.49 2990.53 2993.46 2996.96  2998.2
 2998.88  2999.1 2998.89 2997.52 2996.71 2997.42 2999.18 3001.41 3003.55 3007.16
    2877    2877    2877    2877    2877    2877    2877    2877    2877    2877
    2877    2877    2877    2877    2877    2877    2877    2877    2877    2877
    2877    2877    2877    2877    2877  2925.5  2925.5    2877    2877    2877
    2877    2877    2877    2877    2877    2877    2877    2877    2877    2877
    2877    2877    2877    2877    2877    2877    2877    2877    2877    2877
    2877    2877    2877    2877    2877    2877    2877    2877    2877    2877
Pier Skew, UpSta & Num, DnSta & Num=  ,3805.938, 2 ,3805.938, 2 , 0 , 0 , 0 ,,
       2       2
    2896  2925.5
       2       2
    2896  2925.5
Pier Skew, UpSta & Num, DnSta & Num=  ,3854.429, 2 ,3854.429, 2 , 0 , 0 , 0 ,,
       2       2
    2896  2925.5
       2       2
    2896  2925.5
BR Coef= 1 , 1 , 0 ,1.25, 0 ,,,0.8,0,2,0,
WSPro=,,,, 1 ,,,, 0 ,,,, 0 ,,,,-1 ,-1 ,-1 , 0 , 0 , 0 , 0 , 0
BC Design=,, 0 ,, 0 ,,,,,,
BC HTab HWMax=3010.37

Type RM Length L Ch R = 1 ,23643   ,428,428,428
BEGIN DESCRIPTION:
Little_Rock_Crk_72
END DESCRIPTION:
XS GIS Cut Line= 6
      1067650.86       852775.56      1067637.84       853079.38
      1067807.11       853472.17      1067872.94       853575.28
      1067916.08       853638.86      1067724.64       854019.05
#Sta/Elev= 30
3364.084 2939.483408.515 2931.893491.477 2932.093529.396 2926.373546.862 2927.15
3559.962 2923.863586.926  2922.23621.321 2912.443623.773 2909.46 3624.31 2904.43
3624.463 2907.063625.228 2909.883629.289 2909.043674.638 2922.873687.815  2924.6
3729.947 2918.463786.097 2902.063814.059 2899.143822.562 2896.753858.412 2900.37
3881.317 2919.47 3898.63 2925.55  4063.1 2929.084077.807 2932.184133.959 2972.05
 4149.74 2977.164285.558  2990.44322.559    29984349.754 3007.27  4403.3 3015.13
#Mann= 3 , 0 , 0
3364.084     .06       03814.059     .05       03858.412     .06       0
#XS Ineff= 2 , 0
       03748.095    2928  3921.7       0    2928
Permanent Ineff=
       F       F
Bank Sta=3814.059,3858.412
Skew Angle= 40
Exp/Cntr=0.5,0.3

Type RM Length L Ch R = 1 ,23215   ,582,582,582
BEGIN DESCRIPTION:
little_rock_crk_a8
END DESCRIPTION:
XS GIS Cut Line= 3
      1067654.04       852672.89      1067467.02       853021.75
      1067168.51        853485.7
#Sta/Elev= 30
    4469 2977.67  4502.2 2963.71  4523.8 2955.63  4536.6 2946.84  4554.1 2940.13
  4598.3 2935.99  4636.2 2935.27  4659.8 2932.79  4667.8 2928.38  4685.5 2916.77
  4723.6 2911.96  4744.5  2910.5  4789.5 2909.61  4814.8 2907.62  4878.1 2896.68
    4951 2895.12  4975.6 2892.72  4985.9 2887.61  5014.1 2887.61  5021.8 2889.42
  5038.5 2899.25  5048.8 2908.02    5058 2913.39  5079.9 2931.73    5119  2934.8
  5139.1 2938.08  5150.7 2941.35  5172.9 2945.53  5243.8 2954.52  5416.5 2967.02
#Mann= 4 ,-1 , 0
    4469     .05       0  4975.6     .05       0  5021.8     .09       0
    5119     .05       0
Bank Sta=4975.6,5021.8
Exp/Cntr=0.3,0.1

Type RM Length L Ch R = 1 ,22633   ,651,651,651
BEGIN DESCRIPTION:
Little_Rock_Crk_71
END DESCRIPTION:
XS GIS Cut Line= 2
        1067415.       852400.13      1066690.18       852977.38
#Sta/Elev= 30
  4642.2 3029.03  4676.1 3011.09  4689.2 3002.25  4725.9 2974.26  4749.6 2951.85
  4761.7 2948.74  4787.6 2947.47  4823.7 2924.61    4911 2901.99  4939.2 2896.99
  4959.8 2892.05  4984.5 2880.02  4985.9 2878.79  5014.1 2878.79  5014.4 2880.06
  5109.3 2886.76  5157.8  2890.8  5207.6 2898.73  5257.6 2897.51  5270.2 2893.59
  5270.6 2890.77    5273 2894.65  5279.3 2895.55  5329.8 2897.91    5412 2902.51
  5433.5 2908.26    5451 2910.72  5483.9 2909.44  5528.1 2915.53  5568.8  2917.2
#Mann= 8 ,-1 , 0
  4642.2     .09       0  4823.7     .05       0  4939.2     .08       0
  4984.5     .05       0  5014.4     .08       0  5109.3    .055       0
  5329.8     .09       0    5451     .05       0
Bank Sta=4984.5,5014.4
Exp/Cntr=0.3,0.1

Type RM Length L Ch R = 1 ,21982   ,768,768,768
BEGIN DESCRIPTION:
little_rock_crk_a9
END DESCRIPTION:
XS GIS Cut Line= 2
      1066891.58       851809.73      1066409.65       852568.59
#Sta/Elev= 30
  4542.5 3010.25  4586.9 2996.62  4620.4  2991.9  4661.6 2989.05    4674  2987.1
  4686.8 2978.53  4700.4 2968.08  4710.4 2963.95  4723.1 2962.27  4762.4 2949.98
  4774.9 2948.08  4789.1 2943.21  4850.6 2927.78  4910.5  2909.1  4928.9 2898.33
  4966.3 2873.28  4970.2 2871.03 4977.99 2868.29  4985.1 2865.63  5014.9 2865.63
 5022.18 2867.72  5044.2 2875.51  5141.2 2884.21  5190.8 2886.49  5215.6 2886.53
  5300.3 2890.73  5314.6 2889.97  5339.8 2890.81  5387.5 2889.85  5441.5 2890.17
#Mann= 3 ,-1 , 0
  4542.5     .09       0 4977.99     .05       0 5022.18     .08       0
Bank Sta=4977.99,5022.18
Exp/Cntr=0.3,0.1
